--- CARTER CREEK.prj (project) ---

Proj Title=CARTER CREEK Base Level Engineering
Current Plan=p01
Default Exp/Contr=0.3,0.1
English Units
Geom File=g01
Flow File=f01
Plan File=p01
BEGIN DESCRIPTION:
CARTER CREEK
END DESCRIPTION:

--- CARTER CREEK.p01 (plan) ---

Plan Title=Multiple Run
Short Identifier=Multiple
Geom File=g01
Flow File=f01
Subcritical Flow
K Sum by GR= 0
Std Step Tol= 0.01
Critical Tol= 0.01
Num of Std Step Trials= 20
Max Error Tol= 0.3
Flow Tol Ratio= 0.001
Split Flow NTrial= 30
Split Flow Tol= 0.02
Split Flow Ratio= 0.02
Log Output Level= 0
Friction Slope Method= 1
Unsteady Friction Slope Method= 2
Unsteady Bridges Friction Slope Method= 1
Parabolic Critical Depth
Global Vel Dist=  1 , 1 , 1
Global Log Level= 0
CheckData=True
Encroach Param= -1, 0, 0, 0
BEGIN DESCRIPTION:
Multiple Run
END DESCRIPTION:

--- CARTER CREEK.f01 (steady flow) ---

Flow Title=Multiple
Number of Profiles=7
Profile Names=10-year,25-year,50-year,1pct_min,100-year,1pct_plu,500-year
River Rch & RM= CARTER CREEK,Reach-1,22724
     399     523     622     368     734    1465    1025
River Rch & RM= CARTER CREEK,Reach-1,21225
     557     745     899     539    1075    2146    1542
River Rch & RM= CARTER CREEK,Reach-1,20796
     898    1229    1503     912    1820    3631    2674
River Rch & RM= CARTER CREEK,Reach-1,13223
    1211    1672    2057    1253    2501    4990    3708
River Rch & RM= CARTER CREEK,Reach-1,2562
    1623    2272    2819    1731    3455    6893    5204
Boundary for River Rch & Prof#=CARTER CREEK,Reach-1,1
Up Type=0
Dn Type=3
Dn Slope=0.005
Boundary for River Rch & Prof#=CARTER CREEK,Reach-1,2
Up Type=0
Dn Type=3
Dn Slope=0.005
Boundary for River Rch & Prof#=CARTER CREEK,Reach-1,3
Up Type=0
Dn Type=3
Dn Slope=0.005
Boundary for River Rch & Prof#=CARTER CREEK,Reach-1,4
Up Type=0
Dn Type=3
Dn Slope=0.005
Boundary for River Rch & Prof#=CARTER CREEK,Reach-1,5
Up Type=0
Dn Type=3
Dn Slope=0.005
Boundary for River Rch & Prof#=CARTER CREEK,Reach-1,6
Up Type=0
Dn Type=3
Dn Slope=0.005
Boundary for River Rch & Prof#=CARTER CREEK,Reach-1,7
Up Type=0
Dn Type=3
Dn Slope=0.005

--- CARTER CREEK.g01 (geometry) ---

Geom Title=Existing Conditions

River Reach=CARTER CREEK,Reach-1
Reach XY= 30
      2924457.65      7018436.61      2924181.07      7018253.33
      2923797.95      7017324.13      2923455.59      7017210.71
      2923551.36      7016792.30      2922919.63      7015933.64
      2922883.39      7015386.61      2922602.46      7014741.35
      2922123.38      7014374.32      2921352.77      7014276.12
      2921073.63      7014026.91      2920964.83      7013659.49
      2920404.27      7013292.92      2919355.59      7013780.71
      2918084.92      7013091.47      2917012.50      7013425.32
      2916224.50      7012773.73      2915455.28      7012570.98
      2915036.58      7011985.95      2915164.53      7011091.38
      2914680.14      7010433.55      2914486.31      7009273.79
      2913199.81      7008622.58      2912654.79      7008680.21
      2912269.28      7008133.64      2912311.46      7007552.79
      2912068.68      7007075.66      2911878.57      7007052.23
      2911904.61      7006721.50      2912074.25      7006689.42

Type RM Length L Ch R = 1,22724,116,116,116
BEGIN DESCRIPTION:
CARTER CREEK 39.0
END DESCRIPTION:
XS GIS Cut Line= 3
      2924660.97      7018231.90      2924409.42      7018419.51
      2924246.93      7018630.61
#Sta/Elev= 30
  4686.2  452.74  4729.0  449.58  4735.3  448.44  4742.2  448.47  4749.9  448.44
  4770.7  446.19  4779.1  446.34  4785.3  445.35  4799.9  445.22  4805.6  444.34
  4849.9  442.55  4885.4  439.74  4914.6  438.93  4964.6  439.12  4970.9  439.81
  4993.3  438.91  4999.6  437.79  5003.9  434.89  5004.4  434.09  5009.4  434.09
  5009.9  434.89  5014.3  437.10  5028.4  438.91  5045.6  439.48  5099.5  439.45
  5163.8  441.52  5213.7  444.96  5242.7  448.00  5263.5  448.85  5266.4  449.90
#Mann=6,-1,0
  4686.2     0.1       0  4742.2    0.05       0  4805.6    0.16       0
  5003.9    0.07       0  5009.9    0.16       0  5045.6    0.05       0
Bank Sta=4993.3,5028.4
Exp/Cntr=0.3,0.1

Type RM Length L Ch R = 1,22608,209,209,209
BEGIN DESCRIPTION:
Mapping XS 252a04be
END DESCRIPTION:
XS GIS Cut Line= 3
      2924526.41      7018273.15      2924315.90      7018351.28
      2924250.80      7018559.59
#Sta/Elev= 30
  4779.1  446.96  4797.7  446.52  4803.0  445.69  4822.7  445.00  4828.1  444.29
  4844.6  444.30  4858.4  443.55  4865.9  442.47  4876.6  442.15  4936.1  438.00
  4938.9  437.86  4944.2  438.79  4974.6  439.35  4983.3  437.67  4996.6  432.01
  4997.1  431.21  5002.1  431.21  5002.6  432.01  5018.0  435.63  5023.3  437.42
  5030.7  438.00  5049.5  438.83  5094.9  438.90  5133.3  439.73  5153.3  441.88
  5158.5  444.90  5164.7  446.03  5191.0  445.69  5196.2  446.42  5221.9  446.40
#Mann=4,-1,0
  4779.1    0.16       0  4996.6    0.07       0  5002.6    0.16       0
  5094.9    0.05       0
Bank Sta=4936.1,5030.7
Exp/Cntr=0.3,0.1

Type RM Length L Ch R = 1,22399,263,263,263
BEGIN DESCRIPTION:
Mapping XS 22dfc5e1
END DESCRIPTION:
XS GIS Cut Line= 3
      2924496.01      7018242.77      2924190.03      7018216.73
      2923918.30      7018251.23
#Sta/Elev= 30
  4690.2  448.98  4719.6  447.92  4724.6  448.50  4821.7  440.50  4891.9  438.89
  4902.0  438.45  4912.0  436.71  4922.0  437.10  4932.1  438.73  4938.9  436.37
  4952.2  432.91  4957.9  436.54  4963.0  433.79  4972.2  434.69  4982.3  433.99
  4989.3  431.38  4989.8  430.58  4994.8  430.58  4995.3  431.38  4997.3  431.38
  5002.4  435.18  5006.9  436.37  5012.4  437.84  5020.4  438.43  5025.4  437.50
  5083.0  439.44  5179.1  443.98  5204.0  444.48  5234.2  447.33  5271.2  448.62
#Mann=4,-1,0
  4690.2    0.16       0  4989.3    0.07       0  4995.3    0.16       0
  5179.1    0.05       0
Bank Sta=4938.9,5006.9
Exp/Cntr=0.3,0.1

Type RM Length L Ch R = 1,22136,339,339,339
BEGIN DESCRIPTION:
CARTER CREEK 38.0
END DESCRIPTION:
XS GIS Cut Line= 3
      2924424.96      7017975.00      2924125.00      7017975.00
      2923824.99      7018075.00
#Sta/Elev= 30
  4703.3  452.10  4763.3  449.31  4813.3  447.87  4823.3  446.59  4853.3  445.73
  4913.3  441.07  4953.3  438.99  4963.3  439.24  4973.3  438.66  4983.3  437.62
  4989.1  435.03  4997.8  430.37  4998.3  429.57  5003.3  429.57  5003.8  430.37
  5005.9  430.37  5013.8  435.07  5024.3  436.81  5045.4  436.85  5077.0  433.37
  5079.1  433.63  5087.6  434.67  5108.7  432.56  5119.2  434.61  5125.6  435.03
  5150.8  436.86  5182.5  438.26  5245.7  444.50  5273.4  446.12  5319.5  447.76
#Mann=5,-1,0
  4703.3    0.05       0  4997.8    0.03       0  5003.8    0.05       0
  5079.1    0.16       0  5273.4    0.05       0
Bank Sta=4989.1,5125.6
Exp/Cntr=0.3,0.1

Type RM Length L Ch R = 1,21797,348,348,348
BEGIN DESCRIPTION:
CARTER CREEK 37.0
END DESCRIPTION:
XS GIS Cut Line= 3
      2924224.98      7017675.00      2923925.00      7017725.00
      2923674.98      7017925.02
#Sta/Elev= 30
  4693.5  445.14  4721.4  445.69  4726.4  444.87  4734.0  445.44  4764.4  444.17
  4782.2  442.80  4787.3  441.13  4794.9  440.05  4843.0  436.52  4960.0  433.33
  4977.3  433.48  4987.5  432.86  4995.1  431.31  5000.8  431.31  5001.8  430.49
  5002.3  429.69  5007.3  429.69  5007.8  430.49  5019.2  432.03  5033.6  432.54
  5038.2  433.33  5061.6  434.64  5075.3  436.44  5089.7  437.36  5097.7  438.79
  5118.5  439.81  5132.9  442.10  5139.3  442.03  5161.7  443.79  5317.8  447.99
#Mann=3,-1,0
  4693.5    0.05       0  5001.8    0.03       0  5007.8    0.05       0
Bank Sta=4960,5038.2
Exp/Cntr=0.3,0.1

Type RM Length L Ch R = 1,21449,224,224,224
BEGIN DESCRIPTION:
CARTER CREEK 36.0
END DESCRIPTION:
XS GIS Cut Line= 4
      2924383.16      7017615.60      2923900.00      7017500.00
      2923660.51      7017379.06      2923543.31      7017704.61
#Sta/Elev= 30
  4368.7  449.05  4392.6  446.65  4418.2  447.01  4439.8  442.59  4459.4  443.09
  4500.5  440.26  4719.2  435.64  4767.8  434.70  4786.1  432.97  4871.0  432.09
  4954.7  431.86  4971.4  428.66  4996.3  427.65  4996.8  426.85  5002.3  427.65
  5005.5  429.29  5016.0  430.25  5021.6  431.99  5043.9  432.66  5132.7  431.61
  5241.0  432.97  5277.9  435.93  5283.3  435.43  5299.5  438.21  5331.4  439.84
  5400.8  440.06  5431.5  439.07  5456.9  441.65  5462.2  440.11  5479.8  441.34
#Mann=5,-1,0
  4368.7    0.05       0  4719.2    0.16       0  4871.0    0.05       0
  4996.3    0.03       0  5002.3    0.05       0
Bank Sta=4786.1,5241
Exp/Cntr=0.3,0.1

Type RM Length L Ch R = 1,21225,228,228,228
BEGIN DESCRIPTION:
Mapping XS 7d2c47b4
END DESCRIPTION:
XS GIS Cut Line= 4
      2923874.47      7017285.73      2923749.48      7017271.85
      2923652.25      7017332.61      2923525.53      7017685.00
#Sta/Elev= 30
  4819.6  444.00  4867.9  440.44  4873.0  441.21  4953.8  435.37  4976.4  432.77
  4995.2  431.53  5001.1  426.45  5006.6  426.09  5007.1  425.29  5012.1  425.29
  5012.6  426.09  5016.4  426.24  5022.3  428.83  5031.8  427.95  5037.7  430.44
  5055.8  431.01  5154.1  432.53  5179.5  431.65  5216.3  432.77  5302.4  438.01
  5307.7  437.23  5327.8  437.50  5333.1  436.62  5358.5  438.01  5363.8  436.58
  5389.2  437.81  5394.5  436.91  5419.9  437.93  5425.2  436.88  5434.5  437.27
#Mann=5,-1,0
  4819.6    0.05       0  4953.8    0.16       0  5006.6    0.07       0
  5012.6    0.16       0  5055.8    0.05       0
Bank Sta=4976.4,5216.3
Exp/Cntr=0.3,0.1

Type RM Length L Ch R = 1,20997,201,201,201
BEGIN DESCRIPTION:
Mapping XS 9b360f26
END DESCRIPTION:
XS GIS Cut Line= 4
      2923777.28      7017224.98      2923621.00      7017178.10
      2923560.24      7017209.35      2923492.54      7017730.07
#Sta/Elev= 30
  4772.8  442.19  4823.5  438.70  4837.8  438.55  4856.6  437.41  4861.8  437.82
  4889.7  435.88  4894.9  436.39  4919.6  434.98  4936.0  434.79  4969.9  432.59
  4981.8  432.15  4983.0  432.11  4988.6  428.66  4995.8  427.26  4996.3  426.46
  5001.3  426.46  5001.8  427.26  5010.6  428.44  5020.1  430.77  5069.9  431.29
  5151.2  430.77  5273.1  432.15  5302.4  434.02  5322.6  432.99  5352.9  433.04
  5391.1  434.58  5396.1  434.17  5463.8  435.80  5514.2  435.44  5529.4  436.76
#Mann=7,-1,0
  4772.8    0.05       0  4837.8    0.16       0  4919.6    0.05       0
  4969.9    0.16       0  4995.8    0.07       0  5001.8    0.16       0
  5069.9    0.05       0
Bank Sta=4981.8,5273.1
Exp/Cntr=0.3,0.1

Type RM Length L Ch R = 1,20796,409,409,409
BEGIN DESCRIPTION:
CARTER CREEK 35.0
END DESCRIPTION:
XS GIS Cut Line= 3
      2923924.98      7017225.00      2923475.00      7017125.00
      2923025.02      7017075.00
#Sta/Elev= 30
  4544.2  445.63  4617.2  443.43  4677.3  443.02  4771.4  439.15  4790.6  438.16
  4796.4  437.06  4801.6  437.65  4840.0  435.63  4845.1  436.45  4888.6  434.47
  4893.8  435.41  4913.0  434.61  4932.2  431.55  4937.3  431.87  4943.3  431.02
  4985.9  429.73  4991.8  425.42  4992.3  424.62  4997.6  424.62  4998.1  425.42
  5002.6  427.90  5007.7  427.90  5015.2  430.82  5196.3  429.21  5234.3  431.02
  5286.9  434.07  5327.1  438.58  5377.4  441.51  5417.7  444.72  5457.9  446.56
#Mann=5,-1,0
  4544.2    0.05       0  4771.4    0.16       0  4790.6    0.05       0
  4991.8    0.03       0  4998.1    0.05       0
Bank Sta=4943.3,5234.3
Exp/Cntr=0.3,0.1

Type RM Length L Ch R = 1,20387,323,323,323
BEGIN DESCRIPTION:
Mapping XS 00a3e561
END DESCRIPTION:
XS GIS Cut Line= 3
      2924213.05      7016895.57      2923554.19      7016801.82
      2922868.32      7016921.33
#Sta/Elev= 30
  4333.1  448.56  4369.6  447.68  4440.4  448.47  4587.2  445.23  4658.0  441.11
  4745.3  434.04  4839.5  429.68  4896.8  428.51  4977.6  428.66  4992.5  424.40
  4993.0  423.60  4998.4  423.60  4998.9  424.40  5007.9  427.37  5028.2  428.83
  5158.9  427.86  5180.5  428.01  5211.2  429.68  5251.5  432.18  5278.1  435.87
  5283.2  434.31  5322.6  437.86  5332.6  438.31  5337.7  437.49  5342.9  439.00
  5373.3  441.07  5525.6  444.89  5586.5  447.67  5630.5  447.88  5694.8  450.01
#Mann=3,-1,0
  4333.1    0.05       0  4992.5    0.03       0  4998.9    0.05       0
Bank Sta=4839.5,5211.2
Exp/Cntr=0.3,0.1

Type RM Length L Ch R = 1,20064,76,76,76
BEGIN DESCRIPTION:
Mapping XS 4d578e9d
END DESCRIPTION:
XS GIS Cut Line= 3
      2923960.22      7016517.54      2923415.51      7016519.71
      2922632.13      7016524.05
#Sta/Elev= 30
  4448.8  444.85  4514.0  440.65  4584.0  438.12  4624.0  434.58  4654.0  435.09
  4674.0  433.21  4704.0  431.88  4714.0  432.12  4836.3  428.79  4924.0  427.71
  4954.0  426.71  4984.0  427.66  4996.3  427.36  5000.8  424.73  5001.3  423.93
  5006.7  423.93  5007.2  424.73  5024.0  427.76  5064.0  427.13  5178.9  428.79
  5204.0  430.07  5234.0  432.99  5254.0  436.17  5294.0  438.57  5334.0  438.81
  5384.0  437.37  5514.0  440.56  5594.0  444.37  5694.0  446.36  5776.9  448.96
#Mann=3,-1,0
  4448.8    0.08       0  5000.8    0.07       0  5007.2    0.08       0
Bank Sta=4836.3,5178.9
Exp/Cntr=0.3,0.1

Type RM Length L Ch R = 1,19988,711,711,711
BEGIN DESCRIPTION:
Mapping XS a21e5459
END DESCRIPTION:
XS GIS Cut Line= 3
      2924105.63      7016448.09      2923419.85      7016445.92
      2922618.48      7016454.58
#Sta/Elev= 30
  4287.1  459.60  4387.7  454.91  4437.7  450.00  4527.7  445.73  4567.7  441.72
  4597.7  441.47  4627.7  437.71  4667.7  436.46  4727.7  429.50  4747.7  429.28
  4767.7  432.67  4797.7  428.54  4813.3  428.07  4927.7  427.01  4977.8  427.86
  4997.7  426.32  5004.5  424.44  5005.0  423.64  5010.4  423.64  5010.9  424.44
  5027.7  427.49  5037.7  427.73  5127.7  426.77  5197.6  428.07  5297.8  432.45
  5346.5  431.77  5351.5  432.84  5577.8  438.33  5677.8  444.08  5774.3  446.66
#Mann=3,-1,0
  4287.1    0.05       0  5004.5    0.03       0  5010.9    0.05       0
Bank Sta=4813.3,5197.6
Exp/Cntr=0.3,0.1

Type RM Length L Ch R = 1,19277,521,521,521
BEGIN DESCRIPTION:
CARTER CREEK 32.0
END DESCRIPTION:
XS GIS Cut Line= 3
      2923725.00      7015975.00      2922925.00      7015925.00
      2922475.00      7016125.00
#Sta/Elev= 30
  4190.2  448.78  4200.2  446.98  4220.3  445.41  4380.6  441.29  4428.2  438.66
  4530.9  436.13  4581.0  433.75  4611.0  430.86  4661.1  428.03  4746.4  425.36
  4831.4  423.48  4981.7  425.78  4994.5  425.53  4997.5  422.73  4998.0  421.93
  5003.4  421.93  5003.9  422.73  5013.6  425.44  5112.1  423.52  5166.9  423.87
  5199.0  425.36  5255.1  428.65  5272.9  430.81  5341.9  433.68  5376.8  436.39
  5394.6  435.82  5417.9  437.40  5429.5  440.56  5446.6  443.64  5484.2  446.00
#Mann=3,-1,0
  4190.2    0.05       0  4997.5    0.03       0  5003.9    0.05       0
Bank Sta=4746.4,5199
Exp/Cntr=0.3,0.1

Type RM Length L Ch R = 1,18756,513,513,513
BEGIN DESCRIPTION:
CARTER CREEK 31.0
END DESCRIPTION:
XS GIS Cut Line= 3
      2923324.97      7015425.00      2922875.00      7015425.00
      2922524.96      7015725.03
#Sta/Elev= 30
  4561.2  441.02  4591.2  439.36  4601.2  437.53  4611.2  434.35  4621.2  433.45
  4701.2  428.42  4783.0  424.70  4821.2  423.15  4881.2  422.26  4951.2  423.25
  4991.2  424.86  4997.9  419.59  4998.4  418.79  5003.9  418.79  5004.4  419.59
  5008.7  423.47  5018.3  424.00  5061.1  423.02  5131.4  422.45  5145.6  421.72
  5174.2  422.79  5197.3  424.70  5252.1  429.08  5274.0  431.70  5280.6  432.00
  5294.9  434.16  5309.2  435.35  5358.6  436.29  5401.4  439.06  5472.2  438.82
#Mann=3,-1,0
  4561.2    0.05       0  4997.9    0.03       0  5004.4    0.05       0
Bank Sta=4783,5197.3
Exp/Cntr=0.3,0.1

Type RM Length L Ch R = 1,18243,193,193,193
BEGIN DESCRIPTION:
CARTER CREEK 30.0
END DESCRIPTION:
XS GIS Cut Line= 3
      2923372.54      7015129.08      2922675.00      7014975.00
      2922224.99      7015175.00
#Sta/Elev= 30
  4291.4  434.48  4376.3  430.50  4431.3  429.40  4514.0  430.65  4562.8  428.60
  4667.8  426.46  4698.5  427.52  4717.0  426.29  4752.7  424.18  4797.8  422.21
  4913.6  420.84  4986.5  422.46  4995.5  420.39  4999.9  417.76  5000.4  416.96
  5006.5  417.76  5008.5  417.76  5014.6  421.69  5049.5  421.09  5121.3  424.18
  5141.9  425.25  5165.1  428.55  5170.6  428.18  5211.6  432.82  5217.1  432.18
  5254.3  435.18  5365.0  436.69  5408.6  437.54  5451.1  436.83  5498.2  436.97
#Mann=10,-1,0
  4291.4    0.05       0  4376.3    0.16       0  4431.3    0.05       0
  4717.0    0.16       0  4797.8    0.12       0  4999.9    0.07       0
  5006.5    0.12       0  5254.3    0.16       0  5365.0    0.12       0
  5451.1    0.05       0
Bank Sta=4752.7,5121.3
Exp/Cntr=0.3,0.1

Type RM Length L Ch R = 1,18050,474,474,474
BEGIN DESCRIPTION:
Mapping XS 0f35c06a
END DESCRIPTION:
XS GIS Cut Line= 3
      2923280.49      7014459.83      2922655.53      7014754.95
      2922333.47      7015090.86
#Sta/Elev= 30
  4253.9  435.56  4277.1  437.43  4282.7  436.64  4354.0  439.79  4381.6  440.86
  4547.5  438.56  4607.0  436.51  4624.6  436.88  4669.2  435.90  4708.9  433.45
  4720.8  432.50  4757.6  426.80  4788.0  423.86  4824.0  421.32  4885.7  420.25
  4908.5  421.26  4995.0  421.46  4998.5  418.10  4999.0  417.30  5004.8  417.30
  5005.3  418.10  5009.1  418.67  5016.1  421.98  5058.5  420.40  5086.8  421.19
  5120.7  423.86  5235.6  433.82  5287.4  435.63  5327.4  436.71  5410.4  435.94
#Mann=7,-1,0
  4253.9    0.16       0  4354.0    0.12       0  4624.6    0.16       0
  4708.9    0.12       0  4998.5    0.07       0  5005.3    0.12       0
  5287.4    0.16       0
Bank Sta=4788,5120.7
Exp/Cntr=0.3,0.1

Type RM Length L Ch R = 1,17576,489,489,489
BEGIN DESCRIPTION:
CARTER CREEK 29.0
END DESCRIPTION:
XS GIS Cut Line= 3
      2922717.39      7014266.23      2922332.71      7014546.92
      2922275.00      7015074.97
#Sta/Elev= 30
  4523.8  437.38  4552.4  437.43  4575.6  435.31  4581.8  436.73  4596.5  432.48
  4602.6  436.07  4646.7  434.97  4652.8  431.66  4682.2  430.47  4688.4  428.45
  4696.9  428.79  4703.1  427.22  4752.7  429.73  4803.5  428.12  4954.1  427.00
  4960.3  424.21  4973.0  421.44  4989.6  420.38  4995.5  417.83  5004.7  416.68
  5005.2  415.88  5011.6  416.68  5018.2  420.77  5115.4  420.32  5179.1  419.39
  5209.9  421.44  5271.1  427.91  5309.9  431.48  5400.5  435.30  5531.2  436.64
#Mann=6,-1,0
  4523.8    0.05       0  4752.7    0.16       0  5004.7    0.07       0
  5011.6    0.16       0  5115.4    0.12       0  5271.1    0.16       0
Bank Sta=4973,5209.9
Exp/Cntr=0.3,0.1

Type RM Length L Ch R = 1,17087,524,524,524
BEGIN DESCRIPTION:
CARTER CREEK 28.0
END DESCRIPTION:
XS GIS Cut Line= 3
      2922225.02      7013924.97      2921925.00      7014275.00
      2922074.99      7014774.97
#Sta/Elev= 30
  4515.1  457.71  4586.3  455.38  4643.0  453.17  4726.2  445.73  4741.7  444.11
  4791.7  438.10  4828.3  432.64  4921.0  420.06  4940.4  417.99  4954.7  417.45
  4986.6  418.76  4992.6  415.26  4997.9  417.47  5004.0  414.23  5004.5  413.43
  5010.4  413.43  5010.9  414.23  5017.9  418.67  5153.6  416.88  5174.5  417.40
  5258.0  416.96  5272.8  417.07  5299.6  418.90  5320.2  420.06  5344.1  421.54
  5402.5  428.26  5410.3  429.77  5415.5  429.55  5448.5  432.61  5498.1  434.74
#Mann=9,-1,0
  4515.1    0.16       0  4586.3    0.05       0  4726.2    0.12       0
  4741.7    0.16       0  4828.3    0.12       0  5004.0    0.07       0
  5010.9    0.12       0  5299.6    0.16       0  5402.5    0.05       0
Bank Sta=4921,5320.2
Exp/Cntr=0.3,0.1

Type RM Length L Ch R = 1,16563,633,633,633
BEGIN DESCRIPTION:
CARTER CREEK 27.0
END DESCRIPTION:
XS GIS Cut Line= 3
      2921975.03      7013824.97      2921475.00      7014325.00
      2921425.00      7014774.99
#Sta/Elev= 30
  4301.1  451.98  4343.6  449.48  4414.3  443.91  4541.6  431.99  4591.0  429.14
  4668.8  425.52  4716.5  425.23  4782.0  426.62  4903.4  426.76  4923.4  427.19
  4951.6  418.16  4965.8  416.03  4994.1  415.92  5001.3  413.67  5001.8  412.87
  5007.7  412.87  5008.2  413.67  5018.3  414.99  5131.6  418.16  5189.4  419.25
  5199.4  419.92  5209.5  422.02  5249.7  421.78  5287.3  423.05  5310.1  423.47
  5370.5  427.69  5400.6  434.45  5410.7  435.26  5451.0  433.27  5461.0  433.68
#Mann=7,-1,0
  4301.1    0.16       0  4591.0    0.12       0  4716.5    0.07       0
  4903.4    0.12       0  5001.3    0.07       0  5008.2    0.12       0
  5287.3    0.05       0
Bank Sta=4951.6,5131.6
Exp/Cntr=0.3,0.1

Type RM Length L Ch R = 1,15930,390,390,390
BEGIN DESCRIPTION:
CARTER CREEK 26.0
END DESCRIPTION:
XS GIS Cut Line= 3
      2921424.97      7013675.03      2921075.00      7013975.00
      2920975.00      7014424.99
#Sta/Elev= 30
  4605.6  432.70  4647.8  432.03  4697.8  429.11  4762.0  423.42  4768.5  421.07
  4790.0  420.53  4841.6  414.54  4868.4  412.55  4938.7  412.23  4974.3  413.40
  4988.1  409.72  4998.9  408.86  4999.4  408.06  5005.3  408.06  5005.8  408.86
  5010.0  413.26  5069.1  413.42  5085.7  409.92  5090.9  413.85  5107.5  409.61
  5117.8  410.15  5128.0  413.32  5189.6  414.54  5261.2  419.36  5343.1  428.14
  5366.5  429.57  5394.3  431.25  5448.6  431.22  5486.5  432.71  5527.5  432.68
#Mann=5,-1,0
  4605.6    0.12       0  4998.9    0.07       0  5005.8    0.12       0
  5366.5     0.1       0  5448.6    0.16       0
Bank Sta=4841.6,5189.6
Exp/Cntr=0.3,0.1

Type RM Length L Ch R = 1,15540,292,292,292
BEGIN DESCRIPTION:
CARTER CREEK 25.0
END DESCRIPTION:
XS GIS Cut Line= 3
      2921376.19      7013441.60      2920842.38      7013641.23
      2920524.97      7013925.03
#Sta/Elev= 30
  4507.1  429.57  4558.0  426.30  4625.8  424.39  4643.6  422.88  4673.8  424.14
  4786.2  422.75  4860.7  419.45  4927.2  413.35  4960.7  410.85  4985.7  411.91
  5010.2  408.74  5016.0  408.85  5021.3  412.36  5046.2  410.44  5052.9  411.27
  5141.2  411.40  5159.4  408.66  5159.9  407.86  5165.9  407.86  5166.4  408.66
  5169.6  410.87  5183.9  410.20  5212.3  411.84  5226.5  410.52  5252.6  413.35
  5410.4  424.13  5417.9  425.38  5424.6  424.99  5500.6  429.33  5502.8  429.33
#Mann=5,-1,0
  4507.1    0.16       0  4786.2    0.12       0  5159.4    0.07       0
  5166.4    0.12       0  5500.6     0.1       0
Bank Sta=4927.2,5252.6
Exp/Cntr=0.3,0.1

Type RM Length L Ch R = 1,15248,369,369,369
BEGIN DESCRIPTION:
Mapping XS d70c4f1c
END DESCRIPTION:
XS GIS Cut Line= 3
      2920916.15      7012738.49      2920673.11      7013471.96
      2920495.17      7013914.64
#Sta/Elev= 30
  4196.7  431.53  4275.9  428.93  4339.3  428.52  4402.7  430.20  4408.0  431.42
  4503.1  433.56  4534.8  433.35  4572.3  432.29  4635.5  426.32  4661.6  425.13
  4677.1  422.85  4711.2  419.86  4756.7  414.12  4781.3  412.41  4825.3  409.70
  4983.4  411.09  4998.6  408.78  4999.1  407.98  5005.1  407.98  5005.6  408.78
  5015.8  410.26  5048.1  408.84  5113.3  412.41  5213.0  420.08  5222.5  421.71
  5267.4  425.37  5339.1  428.34  5360.7  427.68  5439.6  428.79  5446.5  428.94
#Mann=8,-1,0
  4196.7    0.05       0  4677.1    0.16       0  4711.2    0.12       0
  4998.6    0.07       0  5005.6    0.12       0  5213.0    0.07       0
  5267.4    0.12       0  5439.6     0.1       0
Bank Sta=4781.3,5113.3
Exp/Cntr=0.3,0.1

Type RM Length L Ch R = 1,14879,553,553,553
BEGIN DESCRIPTION:
CARTER CREEK 24.0
END DESCRIPTION:
XS GIS Cut Line= 3
      2920421.54      7012765.40      2920375.00      7013325.00
      2920411.06      7013941.22
#Sta/Elev= 30
  4472.2  428.76  4532.0  424.59  4552.1  424.24  4609.4  420.93  4622.3  419.15
  4652.4  418.77  4762.8  413.56  4875.4  410.17  5003.6  408.28  5036.2  408.79
  5040.2  408.25  5040.7  407.45  5046.7  407.45  5047.3  408.25  5063.8  409.40
  5073.8  408.92  5093.8  409.84  5113.9  408.63  5153.9  409.37  5164.0  410.17
  5194.0  412.11  5289.8  413.97  5294.8  414.65  5394.3  415.35  5473.9  418.26
  5494.5  418.98  5544.6  422.38  5564.6  424.92  5631.3  425.58  5651.0  427.05
#Mann=4,-1,0
  4472.2    0.05       0  5040.2    0.03       0  5047.3    0.05       0
  5473.9     0.1       0
Bank Sta=4875.4,5164
Exp/Cntr=0.3,0.1

Type RM Length L Ch R = 1,14326,239,239,239
BEGIN DESCRIPTION:
CARTER CREEK 23.0
END DESCRIPTION:
XS GIS Cut Line= 3
      2919977.10      7012945.91      2919925.00      7013575.00
      2920087.92      7014090.83
#Sta/Elev= 30
  4382.6  432.28  4522.2  425.95  4582.4  419.37  4642.6  418.41  4709.4  415.52
  4753.0  416.82  4823.2  414.17  4863.3  414.11  4933.6  410.52  4947.0  408.80
  4983.7  406.09  5000.3  403.64  5000.8  402.84  5006.9  402.84  5007.4  403.64
  5016.5  404.34  5024.3  407.89  5202.3  406.90  5234.5  407.01  5256.9  408.80
  5326.2  414.29  5331.5  413.27  5390.9  418.08  5396.2  417.56  5428.5  420.93
  5433.7  420.33  5493.1  424.67  5498.4  424.01  5516.2  425.35  5554.8  426.80
#Mann=5,-1,0
  4382.6    0.05       0  5000.3    0.03       0  5007.4    0.05       0
  5202.3     0.1       0  5516.2    0.05       0
Bank Sta=4947,5256.9
Exp/Cntr=0.3,0.1

Type RM Length L Ch R = 1,14087,355,355,355
BEGIN DESCRIPTION:
Mapping XS 3dc0392d
END DESCRIPTION:
XS GIS Cut Line= 3
      2919751.40      7012977.22      2919692.38      7013581.34
      2919886.83      7014105.65
#Sta/Elev= 30
  4337.2  438.15  4385.2  437.53  4435.4  432.56  4586.2  424.07  4660.8  421.37
  4762.5  416.00  4907.7  410.50  4939.2  408.35  4980.1  406.02  4990.1  407.20
  4995.5  405.25  4997.9  402.83  4998.4  402.03  5004.5  402.03  5005.0  402.83
  5012.1  406.51  5020.5  407.28  5086.8  405.98  5123.5  406.75  5167.7  408.35
  5252.9  414.57  5308.3  417.81  5313.6  417.41  5338.7  419.42  5363.7  420.22
  5369.1  419.63  5394.5  421.82  5399.4  421.11  5438.7  424.17  5503.4  425.59
#Mann=5,-1,0
  4337.2    0.05       0  4997.9    0.03       0  5005.0    0.05       0
  5123.5     0.1       0  5394.5    0.05       0
Bank Sta=4939.2,5167.7
Exp/Cntr=0.3,0.1

Type RM Length L Ch R = 1,13732,509,509,509
BEGIN DESCRIPTION:
CARTER CREEK 22.0
END DESCRIPTION:
XS GIS Cut Line= 3
      2919379.88      7013171.64      2919425.46      7013781.14
      2919758.35      7014258.41
#Sta/Elev= 30
  4388.8  422.22  4482.4  416.98  4521.0  413.24  4645.2  408.16  4773.2  405.81
  4960.4  406.06  4993.8  406.09  4999.4  401.66  5005.8  401.38  5006.3  400.58
  5012.4  400.58  5012.9  401.38  5016.9  405.85  5188.2  406.55  5218.1  408.16
  5361.0  420.77  5390.6  422.62  5405.5  423.25  5462.2  421.58  5494.4  421.62
  5497.9  422.15  5512.8  420.50  5518.9  421.29  5527.6  420.51  5533.7  421.63
  5548.5  419.67  5557.5  422.17  5563.4  422.95  5569.5  425.53  5581.9  426.88
#Mann=6,-1,0
  4388.8    0.05       0  4960.4    0.16       0  5005.8    0.07       0
  5012.9    0.16       0  5494.4    0.05       0  5557.5    0.16       0
Bank Sta=4645.2,5218.1
Exp/Cntr=0.3,0.1

Type RM Length L Ch R = 1,13223,586,586,586
BEGIN DESCRIPTION:
CARTER CREEK 21.0
END DESCRIPTION:
XS GIS Cut Line= 3
      2919174.99      7013125.03      2918975.00      7013575.00
      2918925.00      7014025.02
#Sta/Elev= 30
  4474.7  432.80  4627.9  427.13  4639.5  425.09  4657.3  424.46  4662.8  423.23
  4680.5  422.10  4761.2  412.40  4855.3  407.08  4877.5  406.60  4883.0  405.71
  4924.4  405.38  4945.2  405.65  4952.8  405.04  4958.2  402.98  4969.6  403.27
  4983.1  401.04  4983.8  400.24  4990.6  400.24  4991.3  401.04  4997.3  401.14
  5017.4  405.52  5087.9  405.10  5124.4  407.08  5148.2  409.09  5222.1  410.36
  5248.8  411.44  5289.1  415.18  5319.3  416.04  5359.5  421.01  5419.9  424.41
#Mann=5,-1,0
  4474.7    0.05       0  4924.4    0.16       0  4983.1    0.07       0
  4991.3    0.16       0  5222.1    0.05       0
Bank Sta=4855.3,5124.4
Exp/Cntr=0.3,0.1

Type RM Length L Ch R = 1,12637,496,496,496
BEGIN DESCRIPTION:
CARTER CREEK 20.0
END DESCRIPTION:
XS GIS Cut Line= 3
      2919074.99      7012975.01      2918575.00      7013275.00
      2918524.99      7013725.05
#Sta/Elev= 30
  4403.3  432.72  4453.8  430.53  4496.6  425.16  4506.3  423.32  4512.1  423.06
  4527.7  420.48  4564.6  416.52  4591.8  411.68  4622.9  408.72  4636.5  406.74
  4651.8  405.82  4694.8  404.32  4803.7  404.38  4862.0  403.87  4877.5  403.08
  4988.9  404.51  4992.3  402.02  4993.0  401.22  4999.8  401.22  5000.5  402.02
  5016.6  404.10  5056.8  403.97  5115.2  405.82  5157.4  409.00  5207.7  415.19
  5217.8  416.97  5308.4  422.74  5348.6  423.14  5409.0  425.03  5439.2  424.52
#Mann=3,-1,0
  4403.3    0.05       0  4992.3    0.03       0  5000.5    0.05       0
Bank Sta=4651.8,5115.2
Exp/Cntr=0.3,0.1

Type RM Length L Ch R = 1,12141,521,521,521
BEGIN DESCRIPTION:
CARTER CREEK 19.0
END DESCRIPTION:
XS GIS Cut Line= 3
      2918434.55      7012480.27      2918125.00      7013075.00
      2918403.30      7013698.98
#Sta/Elev= 30
  4299.4  423.31  4354.0  419.45  4392.6  419.23  4442.4  414.98  4663.8  405.26
  4740.6  403.19  4895.3  402.29  4915.9  403.04  4961.6  402.27  4972.6  401.52
  4974.6  399.37  4975.3  398.57  4982.8  399.37  5007.4  401.22  5013.7  402.98
  5024.6  401.99  5053.9  402.46  5098.8  405.26  5134.5  408.70  5204.2  413.01
  5227.4  415.98  5250.6  417.24  5303.2  417.49  5429.7  423.90  5506.4  424.93
  5561.1  423.71  5597.7  424.82  5620.9  424.34  5644.1  422.33  5653.1  423.02
#Mann=5,-1,0
  4299.4    0.05       0  4915.9    0.16       0  4974.6    0.07       0
  4982.8    0.16       0  5303.2    0.05       0
Bank Sta=4663.8,5098.8
Exp/Cntr=0.3,0.1

Type RM Length L Ch R = 1,11620,576,576,576
BEGIN DESCRIPTION:
CARTER CREEK 18.0
END DESCRIPTION:
XS GIS Cut Line= 3
      2917524.98      7012824.95      2917675.00      7013275.00
      2917475.01      7013724.97
#Sta/Elev= 30
  4550.0  431.60  4592.2  430.87  4602.8  429.67  4655.5  427.57  4666.0  426.40
  4782.0  421.85  4813.6  419.10  4824.1  416.69  4845.2  414.77  4853.3  413.14
  4887.4  408.05  4908.4  406.62  4924.6  404.61  4949.1  400.16  4957.3  399.64
  4999.1  399.50  4999.9  398.70  5006.8  398.70  5007.5  399.50  5061.9  399.77
  5079.1  400.60  5085.3  402.34  5183.8  403.88  5297.9  404.61  5352.0  409.46
  5363.6  412.05  5386.2  415.35  5404.0  415.75  5462.1  421.15  5516.8  422.24
#Mann=7,-1,0
  4550.0    0.05       0  4853.3    0.16       0  4949.1    0.05       0
  4957.3    0.16       0  4999.1    0.07       0  5007.5    0.16       0
  5061.9    0.05       0
Bank Sta=4924.6,5297.9
Exp/Cntr=0.3,0.1

Type RM Length L Ch R = 1,11044,456,456,456
BEGIN DESCRIPTION:
CARTER CREEK 17.0
END DESCRIPTION:
XS GIS Cut Line= 3
      2917424.99      7012975.02      2917175.00      7013375.00
      2916874.97      7013725.04
#Sta/Elev= 30
  4469.0  427.31  4519.1  424.54  4571.0  418.96  4592.2  418.43  4623.7  414.07
  4665.3  409.68  4686.5  409.29  4723.1  405.70  4744.3  406.11  4759.7  404.22
  4814.1  403.45  4890.6  400.17  4997.2  400.15  5007.2  392.80  5008.0  392.00
  5015.7  392.80  5025.7  396.55  5032.9  401.17  5046.6  399.71  5054.3  401.13
  5068.5  400.98  5075.1  399.46  5097.1  402.31  5138.3  403.45  5273.8  406.66
  5281.5  408.65  5309.5  410.06  5327.5  412.68  5373.7  420.10  5401.7  422.97
#Mann=5,-1,0
  4469.0    0.05       0  4623.7    0.16       0  5007.2    0.07       0
  5015.7    0.16       0  5327.5    0.05       0
Bank Sta=4814.1,5138.3
Exp/Cntr=0.3,0.1

Type RM Length L Ch R = 1,10588,668,668,668
BEGIN DESCRIPTION:
CARTER CREEK 16.0
END DESCRIPTION:
XS GIS Cut Line= 3
      2916875.00      7012775.01      2916725.00      7013225.00
      2916675.00      7013675.00
#Sta/Elev= 30
  4465.9  428.53  4560.8  429.76  4634.5  427.67  4666.2  424.22  4740.0  410.55
  4782.1  405.78  4823.6  402.76  4877.0  398.60  4887.5  396.06  4908.6  392.79
  4919.1  392.73  4937.6  400.18  4963.1  400.73  4980.5  400.67  4990.5  397.04
  4996.3  392.49  4997.0  391.69  5004.1  391.69  5004.9  392.49  5010.7  392.64
  5020.7  397.69  5030.8  401.65  5037.1  402.76  5081.1  407.40  5131.4  415.63
  5222.0  419.69  5252.1  420.55  5292.4  419.99  5350.6  422.43  5393.0  423.35
#Mann=5,-1,0
  4465.9    0.16       0  4963.1    0.12       0  4996.3    0.07       0
  5004.9    0.12       0  5350.6    0.05       0
Bank Sta=4823.6,5037.1
Exp/Cntr=0.3,0.1

Type RM Length L Ch R = 1,9920,513,513,513
BEGIN DESCRIPTION:
CARTER CREEK 15.0
END DESCRIPTION:
XS GIS Cut Line= 3
      2916824.99      7012775.00      2916325.00      7012875.00
      2916224.99      7013325.03
#Sta/Elev= 30
  4480.0  429.36  4500.4  428.27  4531.0  424.93  4582.0  416.15  4612.6  412.03
  4638.1  410.03  4704.3  405.17  4724.7  402.72  4764.8  401.82  4796.1  401.80
  4908.3  398.85  4959.3  399.37  4969.5  394.87  4979.7  393.79  4987.3  397.49
  4992.5  397.49  5000.1  394.93  5004.8  392.18  5005.6  391.38  5012.7  391.38
  5013.4  392.18  5030.9  397.56  5059.4  399.82  5103.0  401.82  5143.6  403.08
  5184.5  406.29  5235.7  414.87  5307.5  419.51  5383.0  421.43  5450.9  420.65
#Mann=5,-1,0
  4480.0    0.16       0  4638.1    0.12       0  5004.8    0.07       0
  5013.4    0.12       0  5059.4    0.16       0
Bank Sta=4764.8,5103
Exp/Cntr=0.3,0.1

Type RM Length L Ch R = 1,9407,519,519,519
BEGIN DESCRIPTION:
CARTER CREEK 14.0
END DESCRIPTION:
XS GIS Cut Line= 3
      2916125.02      7012274.96      2915875.00      7012675.00
      2916104.40      7013350.89
#Sta/Elev= 30
  4500.9  427.10  4556.6  423.24  4639.5  417.47  4682.0  413.23  4697.3  412.71
  4718.5  410.00  4751.8  407.99  4784.0  403.88  4828.2  401.45  4834.1  401.86
  4845.0  400.63  4930.9  397.92  4975.3  397.22  4983.1  395.10  4988.3  396.85
  4989.4  390.94  4990.2  390.14  4997.3  390.14  4998.1  390.94  5014.5  397.43
  5121.8  400.19  5132.2  400.63  5176.7  402.08  5239.5  405.88  5265.6  410.65
  5270.9  410.44  5289.5  413.40  5391.2  418.10  5542.9  420.60  5686.4  417.18
#Mann=7,-1,0
  4500.9    0.16       0  4556.6    0.05       0  4751.8    0.16       0
  4930.9    0.12       0  4989.4    0.07       0  4998.1    0.12       0
  5121.8    0.16       0
Bank Sta=4845,5132.2
Exp/Cntr=0.3,0.1

Type RM Length L Ch R = 1,8888,590,590,590
BEGIN DESCRIPTION:
CARTER CREEK 13.0
END DESCRIPTION:
XS GIS Cut Line= 3
      2915775.00      7012225.00      2915425.00      7012525.00
      2915075.03      7012874.97
#Sta/Elev= 30
  4534.4  421.01  4633.7  416.77  4654.6  416.87  4711.7  413.42  4725.9  411.67
  4775.3  408.05  4783.0  406.83  4789.6  406.98  4797.3  405.21  4803.8  404.76
  4818.1  401.51  4840.0  399.18  4846.7  398.27  4875.2  397.13  4910.7  396.99
  4924.6  397.47  4988.2  396.75  4998.9  396.21  5009.5  392.47  5019.3  391.68
  5020.1  390.88  5027.3  390.88  5028.1  391.68  5037.8  395.05  5066.1  396.42
  5122.7  397.35  5171.9  399.18  5334.8  406.91  5363.1  409.44  5490.3  423.88
#Mann=4,-1,0
  4534.4    0.05       0  4910.7    0.16       0  5019.3    0.07       0
  5028.1    0.16       0
Bank Sta=4840,5171.9
Exp/Cntr=0.3,0.1

Type RM Length L Ch R = 1,8298,451,451,451
BEGIN DESCRIPTION:
CARTER CREEK 12.0
END DESCRIPTION:
XS GIS Cut Line= 3
      2915524.98      7011875.01      2915075.00      7012075.00
      2914775.00      7012425.00
#Sta/Elev= 30
  4512.8  420.70  4556.5  419.02  4573.6  415.88  4648.9  409.04  4672.1  405.16
  4677.6  406.13  4695.4  403.48  4700.9  404.61  4718.6  401.71  4741.9  399.76
  4747.4  400.42  4766.3  397.74  4817.1  394.41  4848.0  394.37  4983.3  395.45
  4996.3  394.54  5002.5  390.38  5007.9  389.58  5008.7  388.78  5016.8  389.58
  5018.9  392.71  5033.2  395.82  5069.4  397.27  5073.8  397.74  5104.5  399.26
  5182.5  410.80  5246.1  416.42  5288.9  418.36  5352.6  423.70  5466.2  426.86
#Mann=5,-1,0
  4512.8    0.05       0  4848.0    0.16       0  5007.9    0.07       0
  5016.8    0.16       0  5069.4    0.05       0
Bank Sta=4766.3,5073.8
Exp/Cntr=0.3,0.1

Type RM Length L Ch R = 1,7847,70,70,70
BEGIN DESCRIPTION:
Mapping XS f576bc4a
END DESCRIPTION:
XS GIS Cut Line= 3
      2915731.01      7011711.15      2915184.12      7011685.10
      2914650.27      7011691.61
#Sta/Elev= 30
  4440.5  431.61  4463.1  429.64  4468.1  429.88  4586.7  424.93  4666.8  420.78
  4678.3  419.85  4756.9  410.48  4837.0  399.53  4881.4  396.63  4944.4  394.51
  4990.1  392.59  4992.7  390.12  4993.5  389.32  5000.8  389.32  5001.6  390.12
  5007.1  390.29  5017.9  392.71  5027.1  393.94  5037.1  394.42  5061.6  394.77
  5107.1  395.57  5134.4  396.63  5187.1  399.13  5267.1  406.26  5287.2  409.43
  5337.2  412.58  5385.9  414.55  5390.9  413.78  5407.2  414.79  5521.9  417.46
#Mann=6,-1,0
  4440.5    0.05       0  4944.4    0.08       0  4992.7    0.07       0
  5001.6    0.08       0  5017.9    0.16       0  5061.6    0.05       0
Bank Sta=4881.4,5134.4
Exp/Cntr=0.3,0.1

Type RM Length L Ch R = 1,7777,599,599,599
BEGIN DESCRIPTION:
Mapping XS fb1bc556
END DESCRIPTION:
XS GIS Cut Line= 3
      2915876.44      7011600.47      2915221.02      7011615.66
      2914639.72      7011613.49
#Sta/Elev= 30
  4297.1  442.85  4328.5  440.56  4367.1  436.01  4438.6  432.19  4548.6  429.11
  4664.4  423.22  4688.6  421.86  4718.7  417.69  4748.7  415.16  4828.7  403.52
  4868.7  399.37  4912.1  396.45  4958.7  394.65  4968.7  391.76  4978.7  392.30
  4988.7  387.95  4994.3  387.53  4995.1  386.73  5003.2  387.53  5008.7  391.06
  5018.7  393.87  5159.9  396.17  5168.5  396.46  5188.7  399.00  5218.7  406.83
  5238.7  409.30  5357.9  414.37  5418.7  416.35  5457.0  416.30  5534.0  418.08
#Mann=8,-1,0
  4297.1    0.08       0  4367.1    0.05       0  4664.4    0.08       0
  4994.3    0.07       0  5003.2    0.08       0  5159.9    0.05       0
  5357.9    0.08       0  5457.0    0.05       0
Bank Sta=4912.1,5168.5
Exp/Cntr=0.3,0.1

Type RM Length L Ch R = 1,7178,492,492,492
BEGIN DESCRIPTION:
CARTER CREEK 10.0
END DESCRIPTION:
XS GIS Cut Line= 3
      2915925.02      7011175.00      2915125.00      7011075.00
      2914725.04      7011324.98
#Sta/Elev= 30
  4229.4  452.96  4330.2  441.82  4400.7  437.13  4438.1  431.08  4509.1  421.65
  4582.1  416.47  4612.4  415.66  4642.6  409.89  4743.4  409.86  4750.9  407.46
  4799.5  400.55  4813.9  398.21  4854.1  395.28  4955.0  391.47  4975.2  392.65
  4985.3  390.97  4988.3  385.61  4989.2  384.81  4997.3  385.61  4997.9  390.60
  5005.4  385.97  5015.5  386.24  5033.1  392.10  5043.3  391.60  5079.6  395.28
  5134.4  405.42  5180.1  410.68  5216.7  412.15  5363.5  414.40  5507.3  416.72
#Mann=7,-1,0
  4229.4    0.05       0  4438.1    0.16       0  4799.5    0.12       0
  4988.3    0.07       0  4997.3    0.12       0  5134.4    0.16       0
  5363.5    0.05       0
Bank Sta=4854.1,5079.6
Exp/Cntr=0.3,0.1

Type RM Length L Ch R = 1,6686,534,534,534
BEGIN DESCRIPTION:
CARTER CREEK 9.0
END DESCRIPTION:
XS GIS Cut Line= 3
      2915225.03      7010324.97      2914925.00      7010675.00
      2914625.00      7011025.00
#Sta/Elev= 30
  4529.1  424.16  4628.5  421.60  4677.2  419.19  4720.7  417.72  4777.7  413.58
  4876.5  402.47  4936.4  394.06  4954.4  391.63  4976.4  391.87  4993.4  390.58
  4999.3  384.18  5000.1  383.38  5008.4  384.18  5011.5  388.71  5025.8  391.26
  5075.2  390.53  5163.3  394.06  5164.2  394.11  5224.4  396.14  5245.3  397.99
  5277.3  404.77  5284.7  406.61  5294.7  409.88  5302.4  410.66  5309.0  413.61
  5330.9  412.86  5351.8  410.22  5366.0  410.06  5441.1  414.69  5451.1  415.10
#Mann=8,-1,0
  4529.1    0.16       0  4677.2    0.12       0  4999.3    0.07       0
  5008.4    0.12       0  5164.2    0.16       0  5277.3    0.12       0
  5284.7    0.16       0  5441.1    0.05       0
Bank Sta=4936.4,5163.3
Exp/Cntr=0.3,0.1

Type RM Length L Ch R = 1,6152,540,540,540
BEGIN DESCRIPTION:
CARTER CREEK 8.0
END DESCRIPTION:
XS GIS Cut Line= 3
      2915074.96      7010225.00      2914625.00      7010275.00
      2914275.01      7010574.99
#Sta/Elev= 30
  4558.1  418.78  4632.4  412.20  4739.2  397.80  4789.5  394.00  4823.7  392.66
  4950.5  388.22  4980.6  390.03  4990.7  389.18  5003.8  383.20  5004.6  382.40
  5012.0  382.40  5012.9  383.20  5014.1  383.20  5018.0  389.49  5041.6  392.66
  5046.5  393.97  5053.1  394.33  5060.8  396.83  5067.4  397.26  5075.0  400.59
  5081.6  400.70  5089.3  403.93  5095.9  404.07  5110.2  407.44  5136.1  408.90
  5210.1  413.49  5308.8  413.16  5372.5  415.14  5415.3  414.98  5471.8  416.13
#Mann=6,-1,0
  4558.1    0.16       0  4632.4    0.12       0  5003.8    0.07       0
  5012.9    0.12       0  5136.1    0.16       0  5210.1    0.05       0
Bank Sta=4823.7,5041.6
Exp/Cntr=0.3,0.1

Type RM Length L Ch R = 1,5612,590,590,590
BEGIN DESCRIPTION:
CARTER CREEK 7.0
END DESCRIPTION:
XS GIS Cut Line= 3
      2915024.96      7009575.01      2914475.00      7009775.00
      2914124.98      7010075.02
#Sta/Elev= 30
  4443.4  434.64  4489.2  430.38  4519.8  425.02  4545.1  418.55  4566.3  415.94
  4587.2  413.08  4631.6  405.71  4662.2  402.41  4667.5  403.28  4722.6  399.21
  4779.2  393.91  4852.5  390.73  4921.5  387.76  4988.0  388.25  5002.7  385.66
  5003.6  384.86  5011.9  385.66  5013.3  387.30  5018.6  388.46  5050.0  387.37
  5088.5  388.49  5130.2  390.73  5163.0  394.55  5199.3  402.98  5218.7  405.69
  5241.0  407.77  5298.0  409.75  5328.5  408.87  5470.1  411.95  5489.6  412.42
#Mann=10,-1,0
  4443.4    0.16       0  4566.3    0.12       0  4587.2    0.16       0
  4722.6    0.12       0  5002.7    0.07       0  5011.9    0.12       0
  5088.5    0.16       0  5218.7    0.12       0  5328.5    0.16       0
  5470.1    0.05       0
Bank Sta=4852.5,5130.2
Exp/Cntr=0.3,0.1

Type RM Length L Ch R = 1,5022,602,602,602
BEGIN DESCRIPTION:
CARTER CREEK 6.0
END DESCRIPTION:
XS GIS Cut Line= 3
      2915074.96      7009424.99      2914425.00      7009225.00
      2913924.96      7009575.03
#Sta/Elev= 30
  4332.4  440.31  4374.2  434.20  4414.1  425.31  4452.0  420.64  4484.7  413.78
  4517.4  410.61  4620.7  405.78  4658.7  408.30  4686.1  406.12  4691.4  407.38
  4724.0  405.39  4756.7  401.21  4762.0  402.20  4822.1  393.65  4827.4  394.51
  4874.7  390.26  4885.8  389.33  4939.1  386.63  4958.2  383.66  4963.4  386.36
  4970.6  383.94  4997.4  383.33  4998.2  382.53  5006.6  383.33  5034.7  387.14
  5264.0  385.60  5401.8  389.33  5545.6  402.73  5594.4  408.07  5622.8  409.17
#Mann=6,-1,0
  4332.4    0.16       0  4874.7    0.12       0  4939.1    0.16       0
  4997.4    0.07       0  5006.6    0.16       0  5545.6    0.05       0
Bank Sta=4885.8,5401.8
Exp/Cntr=0.3,0.1

Type RM Length L Ch R = 1,4420,568,568,568
BEGIN DESCRIPTION:
CARTER CREEK 5.0
END DESCRIPTION:
XS GIS Cut Line= 3
      2914275.00      7008525.00      2913975.00      7008975.00
      2913875.01      7009524.96
#Sta/Elev= 30
  4464.5  416.66  4631.3  404.25  4703.4  396.38  4759.4  388.25  4802.5  384.44
  4847.6  384.01  4868.6  385.51  4874.6  383.99  4900.0  383.80  4900.9  383.00
  4908.4  383.00  4909.3  383.80  4910.7  385.33  4919.7  384.96  4933.2  386.78
  5015.5  383.97  5203.0  388.25  5239.1  389.66  5249.3  390.34  5255.6  391.91
  5269.6  391.79  5289.9  393.61  5461.1  397.93  5503.4  398.15  5513.5  399.13
  5523.7  400.88  5532.6  405.29  5537.7  405.17  5544.0  407.81  5564.3  408.82
#Mann=4,-1,0
  4464.5    0.16       0  4900.0    0.07       0  4909.3    0.16       0
  5461.1    0.05       0
Bank Sta=4759.4,5203
Exp/Cntr=0.3,0.1

Type RM Length L Ch R = 1,3852,377,377,377
BEGIN DESCRIPTION:
CARTER CREEK 4.0
END DESCRIPTION:
XS GIS Cut Line= 3
      2914225.01      7008424.99      2913475.00      7008775.00
      2913425.00      7009224.97
#Sta/Elev= 30
  4191.3  416.40  4228.4  414.80  4290.6  409.82  4401.0  399.05  4434.1  397.18
  4490.8  391.78  4581.1  386.84  4724.9  383.75  4787.2  383.40  4875.5  384.40
  4886.2  382.82  4892.9  380.96  4893.8  380.16  4901.4  380.16  4902.2  380.96
  4907.8  381.33  4913.3  383.75  4919.6  384.11  4952.7  383.30  5016.2  386.19
  5051.9  386.84  5097.6  390.89  5129.6  393.41  5210.1  397.77  5240.3  398.56
  5250.4  400.03  5260.4  399.90  5351.0  405.59  5371.1  405.11  5471.7  408.88
#Mann=5,-1,0
  4191.3    0.16       0  4886.2    0.12       0  4892.9    0.07       0
  4902.2    0.12       0  5097.6    0.16       0
Bank Sta=4581.1,5051.9
Exp/Cntr=0.3,0.1

Type RM Length L Ch R = 1,3475,308,308,308
BEGIN DESCRIPTION:
Mapping XS cfbaf946
END DESCRIPTION:
XS GIS Cut Line= 3
      2913410.00      7007990.17      2913178.22      7008513.63
      2913094.93      7009190.35
#Sta/Elev= 30
  4326.7  405.00  4431.9  405.54  4507.0  406.83  4575.9  405.08  4616.3  401.56
  4622.4  400.05  4660.1  396.41  4692.3  391.37  4721.1  388.34  4771.2  385.82
  4819.7  382.99  4882.3  381.93  4930.8  382.66  4936.2  379.17  4937.1  378.37
  4944.7  378.37  4945.6  379.17  4961.0  382.74  4971.3  381.37  4992.3  381.65
  5009.7  385.82  5113.9  395.95  5162.5  398.98  5210.0  399.90  5243.1  402.26
  5291.2  403.53  5377.5  407.90  5484.9  407.80  5515.2  409.24  5581.0  409.95
#Mann=7,-1,0
  4326.7    0.05       0  4431.9    0.16       0  4882.3    0.12       0
  4936.2    0.07       0  4945.6    0.12       0  4992.3    0.16       0
  5113.9    0.05       0
Bank Sta=4771.2,5009.7
Exp/Cntr=0.3,0.1

Type RM Length L Ch R = 1,3167,102,102,102
BEGIN DESCRIPTION:
Mapping XS d70170c3
END DESCRIPTION:
XS GIS Cut Line= 3
      2912787.59      7008195.89      2912844.89      7008547.49
      2913000.90      7009291.16
#Sta/Elev= 30
  4575.9  406.59  4586.0  406.42  4725.6  396.42  4800.8  385.13  4884.5  383.25
  4932.1  381.68  4945.3  377.43  4946.2  376.63  4954.7  377.43  4961.2  382.23
  4984.6  382.77  5093.8  385.13  5200.1  389.73  5215.7  392.45  5245.2  389.23
  5250.4  393.89  5286.0  389.78  5295.1  388.99  5300.3  395.63  5345.0  391.66
  5358.7  396.82  5394.9  391.61  5400.0  397.95  5439.7  393.75  5444.8  400.81
  5489.6  396.08  5494.7  402.18  5589.4  400.17  5594.5  405.04  5692.0  408.34
#Mann=9,-1,0
  4575.9    0.05       0  4586.0    0.08       0  4725.6    0.16       0
  4884.5    0.05       0  4945.3    0.07       0  4954.7    0.05       0
  4984.6    0.08       0  5200.1    0.16       0  5286.0    0.08       0
Bank Sta=4800.8,5093.8
Exp/Cntr=0.3,0.1

Type RM Length L Ch R = 1,3065,503,503,503
BEGIN DESCRIPTION:
CARTER CREEK 3.0
END DESCRIPTION:
XS GIS Cut Line= 3
      2912691.24      7008279.26      2912772.51      7008660.90
      2912881.05      7009251.61
#Sta/Elev= 30
  4609.8  401.23  4651.6  400.25  4656.8  398.02  4677.0  399.48  4687.2  398.75
  4707.7  395.60  4750.8  391.23  4827.4  384.87  4839.7  383.92  4844.8  384.61
  4901.9  382.56  4912.2  381.21  4917.7  377.10  4918.6  376.30  4926.2  376.30
  4927.1  377.10  4934.2  378.33  4938.8  380.42  4953.1  382.00  5034.5  382.86
  5075.3  383.62  5097.5  384.87  5263.1  390.58  5360.0  397.32  5380.4  399.66
  5471.9  405.85  5502.4  405.26  5522.7  407.46  5538.7  408.20  5600.6  409.20
#Mann=5,-1,0
  4609.8    0.08       0  4917.7    0.07       0  4927.1    0.08       0
  4934.2    0.12       0  5034.5    0.08       0
Bank Sta=4827.4,5097.5
Exp/Cntr=0.3,0.1

Type RM Length L Ch R = 1,2562,352,352,352
BEGIN DESCRIPTION:
Mapping XS f13dd043
END DESCRIPTION:
XS GIS Cut Line= 3
      2912696.31      7008357.98      2912503.62      7008396.17
      2911941.09      7008592.36
#Sta/Elev= 30
  4795.3  398.72  4827.2  397.29  4845.6  395.28  4878.2  391.41  4888.4  391.80
  4906.1  388.75  4956.9  383.97  4962.4  383.82  4969.9  381.51  4980.1  380.35
  4988.5  375.18  4994.1  374.60  4995.0  373.80  5004.0  373.80  5004.8  374.60
  5011.5  379.99  5030.5  381.04  5061.6  380.67  5085.6  378.84  5106.8  380.60
  5265.6  381.07  5344.8  383.26  5359.5  383.97  5392.7  386.89  5398.1  388.07
  5477.4  394.47  5548.1  395.74  5553.4  395.06  5579.2  395.76  5587.5  395.17
#Mann=5,-1,0
  4795.3    0.08       0  4845.6    0.12       0  4994.1    0.07       0
  5004.8    0.12       0  5344.8    0.16       0
Bank Sta=4956.9,5359.5
Exp/Cntr=0.3,0.1

Type RM Length L Ch R = 1,2210,455,455,455
BEGIN DESCRIPTION:
CARTER CREEK 2.0
END DESCRIPTION:
XS GIS Cut Line= 3
      2912757.05      7008074.99      2912272.23      7008141.81
      2911875.02      7008374.99
#Sta/Elev= 30
  4510.6  406.25  4522.8  406.68  4542.6  402.40  4549.3  402.63  4573.2  403.15
  4593.4  400.01  4613.6  400.74  4664.1  398.38  4684.3  397.03  4714.6  392.29
  4729.1  391.55  4754.9  390.19  4815.5  384.42  4842.3  383.36  4912.5  380.26
  4984.4  380.24  5000.0  377.51  5003.0  373.81  5003.9  373.01  5012.9  373.01
  5013.7  373.81  5015.2  377.75  5030.9  380.63  5066.4  379.17  5138.9  379.63
  5196.8  381.58  5216.8  383.36  5329.7  395.16  5409.8  405.28  5460.6  408.09
#Mann=6,-1,0
  4510.6    0.16       0  4549.3    0.08       0  4729.1    0.12       0
  5003.0    0.07       0  5013.7    0.12       0  5138.9    0.16       0
Bank Sta=4842.3,5216.8
Exp/Cntr=0.3,0.1

Type RM Length L Ch R = 1,1755,699,699,699
BEGIN DESCRIPTION:
Mapping XS 7450d00e
END DESCRIPTION:
XS GIS Cut Line= 3
      2912788.35      7007932.63      2912302.23      7007759.01
      2911449.00      7008019.15
#Sta/Elev= 30
  4472.8  407.87  4542.5  406.83  4561.3  405.64  4568.2  404.07  4614.4  403.55
  4635.6  400.23  4646.8  400.47  4686.1  397.89  4691.4  399.06  4716.9  395.09
  4778.5  396.97  4809.3  395.12  4921.8  384.60  4927.1  385.05  4944.3  382.39
  4983.4  379.37  4987.5  380.21  4991.9  378.95  4997.1  374.41  5001.7  373.75
  5002.5  372.95  5012.4  373.75  5029.9  379.74  5133.6  379.87  5184.7  378.39
  5237.7  379.91  5290.8  382.39  5576.0  404.19  5686.5  408.01  5881.0  408.98
#Mann=6,-1,0
  4472.8    0.16       0  4542.5    0.08       0  4646.8    0.12       0
  5001.7    0.07       0  5012.4    0.12       0  5237.7    0.16       0
Bank Sta=4944.3,5290.8
Exp/Cntr=0.3,0.1
