--- CEDAR CREEK.prj (project) ---

Proj Title=CEDAR CREEK Base Level Engineering
Current Plan=p01
Default Exp/Contr=0.3,0.1
English Units
Geom File=g01
Flow File=f01
Plan File=p01
BEGIN DESCRIPTION:
CEDAR CREEK
END DESCRIPTION:

--- CEDAR CREEK.p01 (plan) ---

Plan Title=Multiple Run
Short Identifier=Multiple
Geom File=g01
Flow File=f01
Subcritical Flow
K Sum by GR= 0
Std Step Tol= 0.01
Critical Tol= 0.01
Num of Std Step Trials= 20
Max Error Tol= 0.3
Flow Tol Ratio= 0.001
Split Flow NTrial= 30
Split Flow Tol= 0.02
Split Flow Ratio= 0.02
Log Output Level= 0
Friction Slope Method= 1
Unsteady Friction Slope Method= 2
Unsteady Bridges Friction Slope Method= 1
Parabolic Critical Depth
Global Vel Dist=  1 , 1 , 1
Global Log Level= 0
CheckData=True
Encroach Param= -1, 0, 0, 0
BEGIN DESCRIPTION:
Multiple Run
END DESCRIPTION:

--- CEDAR CREEK.f01 (steady flow) ---

Flow Title=Multiple
Number of Profiles=7
Profile Names=10-year,25-year,50-year,1pct_min,100-year,1pct_plu,500-year
River Rch & RM= CEDAR CREEK,Reach-1,57483
     459     597     704     412     823    1642    1121
River Rch & RM= CEDAR CREEK,Reach-1,56804
     860    1155    1394     833    1662    3316    2358
River Rch & RM= CEDAR CREEK,Reach-1,48045
    1398    1926    2362    1432    2858    5702    4178
River Rch & RM= CEDAR CREEK,Reach-1,37587
    1666    2308    2841    1728    3447    6877    5068
River Rch & RM= CEDAR CREEK,Reach-1,28821
    1704    2358    2902    1764    3519    7021    5168
River Rch & RM= CEDAR CREEK,Reach-1,25505
    1933    2692    3327    2029    4048    8077    5989
River Rch & RM= CEDAR CREEK,Reach-1,16642
    2008    2797    3456    2108    4205    8390    6220
River Rch & RM= CEDAR CREEK,Reach-1,11716
    2444    3435    4270    2617    5222   10420    7808
River Rch & RM= CEDAR CREEK,Reach-1,10003
    2638    3719    4632    2845    5676   11325    8517
Boundary for River Rch & Prof#=CEDAR CREEK,Reach-1,1
Up Type=0
Dn Type=3
Dn Slope=0.005
Boundary for River Rch & Prof#=CEDAR CREEK,Reach-1,2
Up Type=0
Dn Type=3
Dn Slope=0.005
Boundary for River Rch & Prof#=CEDAR CREEK,Reach-1,3
Up Type=0
Dn Type=3
Dn Slope=0.005
Boundary for River Rch & Prof#=CEDAR CREEK,Reach-1,4
Up Type=0
Dn Type=3
Dn Slope=0.005
Boundary for River Rch & Prof#=CEDAR CREEK,Reach-1,5
Up Type=0
Dn Type=3
Dn Slope=0.005
Boundary for River Rch & Prof#=CEDAR CREEK,Reach-1,6
Up Type=0
Dn Type=3
Dn Slope=0.005
Boundary for River Rch & Prof#=CEDAR CREEK,Reach-1,7
Up Type=0
Dn Type=3
Dn Slope=0.005

--- CEDAR CREEK.g01 (geometry) ---

Geom Title=Existing Conditions

River Reach=CEDAR CREEK,Reach-1
Reach XY= 30
      2785205.59      7100170.71      2785404.27      7097996.89
      2784822.01      7097060.74      2785279.50      7095313.05
      2785915.56      7094635.71      2785257.96      7090686.45
      2786270.37      7089943.33      2786565.04      7088095.51
      2786268.82      7087451.87      2787972.96      7085339.62
      2787930.24      7084572.39      2788643.17      7083599.35
      2788087.77      7081766.69      2789115.74      7080258.70
      2788446.34      7079341.58      2789189.40      7078875.31
      2788978.10      7077705.18      2789365.46      7077541.29
      2788915.71      7077148.34      2789669.96      7076553.33
      2789973.51      7075443.38      2788921.30      7073050.29
      2788463.17      7073135.03      2788231.31      7072397.54
      2787621.40      7072372.40      2786287.04      7071207.52
      2787041.40      7069245.81      2786669.69      7067608.36
      2785768.31      7066934.87      2786375.59      7065920.71

Type RM Length L Ch R = 1,57483,379,379,379
BEGIN DESCRIPTION:
CEDAR CREEK 71.0
END DESCRIPTION:
XS GIS Cut Line= 3
      2785475.01      7099575.00      2785175.00      7099575.00
      2784575.03      7100074.98
#Sta/Elev= 30
  4721.0  600.47  4731.0  599.65  4751.0  595.42  4781.0  594.03  4871.0  591.04
  4901.0  592.93  4911.0  592.89  4931.0  592.13  4954.8  589.77  4981.0  586.61
  4988.0  583.84  4988.5  583.04  4993.5  583.04  4994.0  583.84  5013.3  589.77
  5018.5  590.39  5085.4  590.91  5092.0  591.74  5120.6  591.08  5149.2  592.15
  5163.6  591.20  5170.1  589.83  5198.7  590.21  5213.0  591.41  5241.7  591.68
  5255.3  592.87  5333.4  593.19  5397.9  595.85  5624.4  597.55  5802.0  600.36
#Mann=3,-1,0
  4721.0    0.05       0  4988.0    0.03       0  4994.0    0.05       0
Bank Sta=4954.8,5013.3
Exp/Cntr=0.3,0.1

Type RM Length L Ch R = 1,57104,300,300,300
BEGIN DESCRIPTION:
CEDAR CREEK 70.0
END DESCRIPTION:
XS GIS Cut Line= 3
      2785574.96      7099274.99      2785275.00      7099225.00
      2784775.01      7099425.00
#Sta/Elev= 30
  4681.3  596.58  4853.6  593.33  4944.9  589.66  4975.3  587.36  4982.9  584.80
  4988.1  584.80  4991.8  583.25  4992.3  582.45  4997.3  582.45  4997.8  583.25
  5000.2  584.39  5006.9  585.37  5017.7  588.25  5022.6  588.45  5060.8  589.18
  5075.1  588.47  5093.1  588.72  5137.5  590.80  5161.8  589.79  5179.3  587.67
  5200.8  588.44  5215.6  588.26  5233.1  589.48  5275.1  589.66  5293.7  590.03
  5317.9  591.40  5347.5  591.17  5377.2  591.64  5401.4  592.95  5523.9  594.27
#Mann=5,-1,0
  4681.3    0.05       0  4991.8    0.03       0  4997.8    0.05       0
  5022.6    0.16       0  5075.1    0.05       0
Bank Sta=4944.9,5275.1
Exp/Cntr=0.3,0.1

Type RM Length L Ch R = 1,56804,370,370,370
BEGIN DESCRIPTION:
CEDAR CREEK 69.0
END DESCRIPTION:
XS GIS Cut Line= 3
      2785524.98      7099174.99      2785075.00      7099025.00
      2784675.02      7099025.00
#Sta/Elev= 30
  4533.1  595.04  4585.8  593.62  4617.4  593.46  4649.0  591.86  4680.6  591.83
  4733.4  590.40  4754.4  590.71  4820.9  589.24  4862.5  588.63  4933.6  587.47
  4975.8  587.72  4986.3  587.04  4993.9  582.57  4994.4  581.77  4999.4  581.77
  4999.9  582.57  5009.9  583.21  5017.4  585.34  5027.4  586.00  5047.4  586.54
  5057.4  587.49  5087.4  587.13  5093.8  587.64  5114.7  589.24  5157.4  589.79
  5192.9  591.31  5317.4  592.69  5357.4  593.97  5387.4  593.92  5407.4  594.54
#Mann=6,-1,0
  4533.1    0.05       0  4862.5    0.12       0  4993.9    0.07       0
  4999.9    0.12       0  5093.8    0.16       0  5192.9    0.05       0
Bank Sta=4820.9,5114.7
Exp/Cntr=0.3,0.1

Type RM Length L Ch R = 1,56434,372,372,372
BEGIN DESCRIPTION:
CEDAR CREEK 68.0
END DESCRIPTION:
XS GIS Cut Line= 3
      2785574.97      7098824.99      2785275.00      7098725.00
      2784875.01      7098775.00
#Sta/Elev= 30
  4680.3  593.59  4764.6  591.54  4796.2  590.21  4827.8  589.75  4848.9  588.86
  4873.0  588.30  4943.8  587.63  4952.9  586.65  4975.4  585.72  4977.7  584.70
  4986.0  581.00  4990.9  580.28  4991.4  579.48  4996.4  579.48  4996.9  580.28
  4999.0  580.28  5016.7  584.24  5026.7  585.51  5057.0  585.77  5077.1  587.40
  5087.2  587.37  5107.4  586.49  5128.3  586.65  5208.1  586.78  5248.4  587.22
  5288.8  588.82  5308.9  589.19  5329.1  590.09  5378.9  591.44  5399.6  591.51
#Mann=6,-1,0
  4680.3    0.05       0  4873.0    0.16       0  4977.7    0.12       0
  4990.9    0.07       0  4996.9    0.12       0  5378.9    0.05       0
Bank Sta=4952.9,5128.3
Exp/Cntr=0.3,0.1

Type RM Length L Ch R = 1,56062,435,435,435
BEGIN DESCRIPTION:
CEDAR CREEK 67.0
END DESCRIPTION:
XS GIS Cut Line= 3
      2785775.02      7098725.01      2785175.00      7098425.00
      2784574.97      7098725.02
#Sta/Elev= 30
  4273.3  597.99  4496.9  592.03  4533.3  589.54  4756.2  585.79  4786.2  585.69
  4921.8  584.41  4941.4  581.96  4966.5  583.52  4973.0  582.69  4988.9  580.98
  4997.3  577.64  5008.2  577.35  5008.7  576.55  5014.2  577.35  5033.6  582.51
  5042.0  580.60  5055.9  582.06  5064.3  583.67  5069.9  586.00  5078.3  587.16
  5100.7  587.11  5109.1  585.22  5114.6  586.76  5123.0  584.80  5139.0  585.03
  5159.8  585.79  5181.9  587.80  5251.1  588.44  5391.4  589.86  5615.0  594.12
#Mann=8,-1,0
  4273.3    0.05       0  4786.2    0.16       0  4973.0    0.12       0
  5008.2    0.07       0  5014.2    0.12       0  5139.0    0.16       0
  5181.9    0.12       0  5251.1    0.05       0
Bank Sta=4756.2,5159.8
Exp/Cntr=0.3,0.1

Type RM Length L Ch R = 1,55627,431,431,431
BEGIN DESCRIPTION:
CEDAR CREEK 66.0
END DESCRIPTION:
XS GIS Cut Line= 3
      2785875.01      7098275.00      2785275.00      7098125.00
      2784674.98      7098375.01
#Sta/Elev= 30
  4390.8  596.44  4442.4  593.01  4720.7  588.44  4757.7  584.47  4803.1  584.17
  4821.2  586.13  4826.3  584.61  4844.4  588.05  4867.5  589.00  4875.3  586.76
  4885.6  585.68  4912.8  585.22  4944.9  584.69  4957.7  583.13  4978.4  583.81
  4991.2  581.09  4996.0  575.59  4996.5  574.79  5002.0  575.59  5006.7  581.09
  5018.5  582.19  5063.4  582.09  5077.0  580.78  5085.1  581.10  5100.8  585.20
  5124.7  583.87  5222.1  584.47  5250.3  585.38  5408.5  588.61  5659.3  591.10
#Mann=5,-1,0
  4390.8    0.05       0  4912.8    0.16       0  4996.0    0.07       0
  5002.0    0.16       0  5250.3    0.05       0
Bank Sta=4757.7,5222.1
Exp/Cntr=0.3,0.1

Type RM Length L Ch R = 1,55196,364,364,364
BEGIN DESCRIPTION:
CEDAR CREEK 65.0
END DESCRIPTION:
XS GIS Cut Line= 3
      2785575.02      7097825.00      2785275.00      7097875.00
      2784874.97      7098225.02
#Sta/Elev= 30
  4693.4  586.80  4734.0  586.18  4754.2  586.78  4764.4  586.27  4777.3  583.51
  4825.2  582.29  4875.9  583.15  4908.8  582.52  4926.6  581.47  4944.7  579.03
  4957.0  579.26  4966.7  580.54  4987.4  580.33  4995.0  577.98  5000.9  577.98
  5001.7  575.09  5002.2  574.29  5007.2  574.29  5007.7  575.09  5011.3  577.78
  5018.9  579.66  5033.1  582.33  5047.4  583.47  5082.5  583.63  5125.2  581.27
  5214.8  582.77  5282.3  583.51  5429.9  586.04  5501.1  589.01  5529.1  589.03
#Mann=6,-1,0
  4693.4    0.05       0  4944.7    0.16       0  4966.7    0.12       0
  5001.7    0.07       0  5007.7    0.12       0  5214.8    0.05       0
Bank Sta=4777.3,5282.3
Exp/Cntr=0.3,0.1

Type RM Length L Ch R = 1,54832,750,750,750
BEGIN DESCRIPTION:
CEDAR CREEK 64.0
END DESCRIPTION:
XS GIS Cut Line= 3
      2785719.17      7097546.93      2785225.00      7097625.00
      2784674.99      7097925.00
#Sta/Elev= 30
  4473.9  588.03  4753.2  584.62  4771.7  586.90  4826.3  582.77  4945.5  582.52
  4980.2  579.90  4997.0  576.41  5001.1  573.10  5001.6  572.30  5007.1  573.10
  5009.8  578.12  5019.8  580.71  5038.7  578.65  5047.8  577.09  5076.7  582.38
  5094.5  581.01  5135.1  582.80  5151.2  578.66  5167.4  579.70  5179.2  583.67
  5208.8  581.02  5234.5  582.28  5260.4  584.09  5270.4  582.23  5299.8  582.77
  5323.1  585.26  5358.2  583.64  5483.5  586.44  5521.0  589.67  5600.7  590.25
#Mann=9,-1,0
  4473.9    0.05       0  4980.2    0.16       0  5001.1    0.07       0
  5007.1    0.16       0  5038.7    0.12       0  5094.5    0.16       0
  5208.8    0.12       0  5234.5    0.16       0  5323.1    0.05       0
Bank Sta=4826.3,5299.8
Exp/Cntr=0.3,0.1

Type RM Length L Ch R = 1,54082,412,412,412
BEGIN DESCRIPTION:
CEDAR CREEK 63.0
END DESCRIPTION:
XS GIS Cut Line= 3
      2786075.03      7097525.01      2784875.00      7097125.00
      2784574.98      7097175.00
#Sta/Elev= 30
  3722.7  594.69  3817.6  592.05  3965.2  589.99  4017.9  590.27  4070.6  587.43
  4260.3  586.12  4439.5  583.88  4481.7  582.41  4566.0  583.10  4587.1  581.62
  4614.7  581.60  4629.2  582.32  4645.3  580.88  4671.4  579.68  4882.2  580.38
  4945.5  579.40  4966.6  576.93  4990.2  576.40  4994.8  570.98  4995.3  570.18
  5000.8  570.98  5007.9  570.99  5015.5  575.15  5038.3  580.29  5049.1  580.88
  5058.6  582.16  5149.8  584.63  5198.0  587.55  5247.8  587.23  5291.8  588.19
#Mann=5,-1,0
  3722.7    0.05       0  4614.7    0.16       0  4994.8    0.07       0
  5000.8    0.16       0  5247.8    0.05       0
Bank Sta=4645.3,5049.1
Exp/Cntr=0.3,0.1

Type RM Length L Ch R = 1,53670,563,563,563
BEGIN DESCRIPTION:
CEDAR CREEK 62.0
END DESCRIPTION:
XS GIS Cut Line= 3
      2786074.99      7097325.00      2784875.00      7096825.00
      2784475.00      7097025.00
#Sta/Elev= 30
  3727.6  594.49  3803.4  591.95  3987.6  589.95  4049.9  587.46  4179.9  586.00
  4238.4  586.71  4286.0  582.58  4333.7  582.58  4355.9  585.16  4377.6  582.60
  4416.0  581.36  4668.2  579.38  4686.4  578.91  4735.1  577.24  4776.8  578.17
  4789.3  575.41  4811.5  579.19  4905.0  578.74  4973.4  578.45  4989.1  574.97
  4992.1  569.80  4992.6  569.00  4998.1  569.80  5005.9  574.49  5024.9  578.51
  5065.9  579.38  5237.2  585.57  5288.6  585.59  5354.6  584.51  5474.8  588.75
#Mann=6,-1,0
  3727.6    0.05       0  4686.4    0.16       0  4905.0    0.12       0
  4992.1    0.07       0  4998.1    0.12       0  5288.6    0.05       0
Bank Sta=4668.2,5065.9
Exp/Cntr=0.3,0.1

Type RM Length L Ch R = 1,53107,504,504,504
BEGIN DESCRIPTION:
CEDAR CREEK 61.0
END DESCRIPTION:
XS GIS Cut Line= 3
      2785542.66      7096656.24      2785254.80      7096569.49
      2784725.05      7096625.00
#Sta/Elev= 30
  4634.3  582.36  4673.6  582.38  4695.2  583.21  4761.2  580.90  4816.3  578.04
  4872.1  575.72  4903.6  577.00  4943.1  577.46  4954.9  577.68  4964.9  576.93
  4995.1  573.28  5002.1  568.58  5002.6  567.78  5007.6  567.78  5008.1  568.58
  5015.2  573.95  5025.2  574.87  5045.3  575.44  5065.5  574.40  5085.6  577.20
  5144.8  578.20  5166.0  577.61  5196.2  578.90  5216.3  577.80  5265.8  578.04
  5316.8  579.68  5371.6  580.21  5387.2  581.38  5409.3  581.17  5467.6  582.74
#Mann=7,-1,0
  4634.3    0.05       0  4943.1    0.12       0  5002.1    0.07       0
  5008.1    0.12       0  5144.8    0.16       0  5371.6    0.12       0
  5409.3    0.16       0
Bank Sta=4816.3,5265.8
Exp/Cntr=0.3,0.1

Type RM Length L Ch R = 1,52603,509,509,509
BEGIN DESCRIPTION:
CEDAR CREEK 60.0
END DESCRIPTION:
XS GIS Cut Line= 3
      2785875.02      7096575.01      2785075.00      7096225.00
      2784599.30      7096256.94
#Sta/Elev= 30
  4118.7  589.04  4127.7  589.62  4133.1  588.84  4156.5  590.15  4173.3  587.92
  4179.9  586.11  4203.3  584.78  4383.4  583.15  4505.8  580.53  4566.2  578.17
  4588.1  578.55  4683.6  576.79  4749.9  576.10  4925.3  575.60  4983.0  573.46
  4994.4  572.68  5002.0  570.60  5009.0  569.96  5009.5  569.16  5014.5  569.16
  5015.0  569.96  5022.0  574.21  5032.0  575.00  5066.8  574.36  5135.0  576.71
  5136.8  576.78  5216.6  579.58  5252.5  577.39  5292.6  580.11  5468.7  582.96
#Mann=5,-1,0
  4118.7    0.05       0  4749.9    0.12       0  5009.0    0.07       0
  5015.0    0.12       0  5135.0    0.16       0
Bank Sta=4683.6,5136.8
Exp/Cntr=0.3,0.1

Type RM Length L Ch R = 1,52094,832,832,832
BEGIN DESCRIPTION:
CEDAR CREEK 59.0
END DESCRIPTION:
XS GIS Cut Line= 3
      2785974.99      7096025.00      2785213.14      7095913.24
      2784589.89      7095959.99
#Sta/Elev= 30
  4197.4  585.07  4288.3  583.93  4366.9  580.68  4490.5  579.46  4621.9  575.72
  4755.2  575.07  4760.0  574.70  4813.9  571.47  4824.0  569.37  4844.2  570.36
  4850.6  574.20  4904.9  574.40  4920.4  575.51  4967.4  574.70  4985.6  571.64
  4992.6  567.31  4993.1  566.51  4998.7  567.31  5005.6  570.79  5015.7  572.68
  5071.2  575.07  5105.9  578.23  5136.0  577.78  5186.2  580.03  5216.2  579.00
  5256.3  580.64  5328.4  580.03  5436.9  581.92  5527.1  580.89  5592.4  582.96
#Mann=5,-1,0
  4197.4    0.05       0  4760.0    0.12       0  4992.6    0.07       0
  4998.7    0.12       0  5136.0    0.16       0
Bank Sta=4755.2,5071.2
Exp/Cntr=0.3,0.1

Type RM Length L Ch R = 1,51262,1233,1233,1233
BEGIN DESCRIPTION:
CEDAR CREEK 58.0
END DESCRIPTION:
XS GIS Cut Line= 3
      2785874.97      7095874.97      2785275.00      7095375.00
      2784824.95      7095324.99
#Sta/Elev= 30
  4222.3  582.62  4286.7  579.33  4676.9  572.44  4741.0  573.79  4825.6  571.74
  4868.8  572.48  4949.0  571.55  4967.5  571.53  4975.3  570.01  4981.8  570.95
  4989.6  567.37  4996.1  567.47  4996.9  562.84  4997.4  562.04  5002.6  562.04
  5003.1  562.84  5005.3  562.84  5023.4  568.90  5033.5  570.99  5053.6  571.77
  5073.7  569.78  5093.8  569.77  5104.1  572.44  5114.0  574.41  5119.6  574.43
  5224.6  576.33  5264.9  572.83  5295.1  576.10  5325.3  577.21  5456.1  579.20
#Mann=7,-1,0
  4222.3    0.05       0  4868.8    0.12       0  4949.0    0.16       0
  4996.9    0.07       0  5003.1    0.16       0  5005.3    0.12       0
  5119.6    0.16       0
Bank Sta=4676.9,5104.1
Exp/Cntr=0.3,0.1

Type RM Length L Ch R = 1,50029,521,521,521
BEGIN DESCRIPTION:
CEDAR CREEK 57.0
END DESCRIPTION:
XS GIS Cut Line= 3
      2786324.98      7094825.00      2785875.00      7094725.00
      2784874.96      7094925.01
#Sta/Elev= 30
  4551.6  577.93  4654.0  574.83  4711.6  571.57  4755.2  571.64  4760.3  573.23
  4803.8  570.06  4869.1  570.74  4880.9  569.56  4896.0  566.64  4920.4  569.64
  4961.3  569.39  4981.8  567.09  4988.2  565.08  4993.4  565.48  5004.7  562.72
  5006.8  562.67  5007.3  561.87  5013.1  562.67  5015.1  562.67  5022.8  567.61
  5033.0  568.53  5303.4  569.56  5309.2  569.60  5410.7  570.87  5532.7  574.92
  5583.6  573.77  5634.6  575.78  5657.7  575.02  5736.6  574.53  6032.4  578.01
#Mann=7,-1,0
  4551.6    0.05       0  5004.7    0.16       0  5006.8    0.03       0
  5013.1    0.16       0  5309.2    0.12       0  5410.7    0.16       0
  5657.7    0.05       0
Bank Sta=4880.9,5303.4
Exp/Cntr=0.3,0.1

Type RM Length L Ch R = 1,49508,565,565,565
BEGIN DESCRIPTION:
CEDAR CREEK 56.0
END DESCRIPTION:
XS GIS Cut Line= 3
      2786582.93      7094631.99      2785825.00      7094275.00
      2784832.91      7094329.91
#Sta/Elev= 30
  4147.7  581.22  4225.5  579.75  4255.9  577.45  4385.1  577.20  4590.9  570.95
  4664.0  570.73  4687.2  568.97  4695.0  568.80  4749.1  567.48  4910.8  567.64
  4988.0  567.33  5002.4  560.67  5002.9  559.87  5008.7  560.67  5015.5  566.67
  5025.6  567.28  5125.7  566.28  5145.7  564.54  5165.8  568.37  5194.1  568.80
  5215.0  570.04  5296.0  572.82  5406.1  572.40  5446.2  573.78  5526.9  572.32
  5596.4  571.26  5620.1  572.61  5636.5  571.66  5915.5  575.46  5979.1  575.98
#Mann=10,-1,0
  4147.7    0.05       0  4590.9    0.16       0  4687.2    0.05       0
  4749.1    0.16       0  4910.8    0.12       0  5002.4    0.07       0
  5008.7    0.12       0  5215.0    0.05       0  5526.9    0.16       0
  5915.5    0.05       0
Bank Sta=4695,5194.1
Exp/Cntr=0.3,0.1

Type RM Length L Ch R = 1,48943,435,435,435
BEGIN DESCRIPTION:
CEDAR CREEK 55.0
END DESCRIPTION:
XS GIS Cut Line= 3
      2786681.89      7093902.83      2785875.00      7093775.00
      2784942.31      7093845.54
#Sta/Elev= 30
  4178.6  574.77  4307.1  572.94  4357.7  570.71  4499.4  570.13  4529.8  567.98
  4763.7  565.56  4872.6  564.38  4914.6  565.17  4934.8  563.19  4955.1  564.96
  4985.4  564.84  5012.4  562.34  5012.9  561.54  5018.8  562.34  5025.6  564.35
  5058.1  565.56  5085.8  567.83  5102.8  566.68  5156.0  566.46  5176.1  568.26
  5236.2  569.09  5276.3  567.61  5346.5  568.84  5376.6  571.15  5426.8  571.18
  5455.8  569.50  5537.1  570.33  5600.2  568.51  5717.6  568.16  5930.9  572.41
#Mann=6,-1,0
  4178.6    0.05       0  4872.6    0.12       0  5012.4    0.07       0
  5018.8    0.12       0  5102.8    0.05       0  5600.2    0.16       0
Bank Sta=4763.7,5058.1
Exp/Cntr=0.3,0.1

Type RM Length L Ch R = 1,48508,463,463,463
BEGIN DESCRIPTION:
CEDAR CREEK 54.0
END DESCRIPTION:
XS GIS Cut Line= 3
      2787425.03      7093675.01      2785875.00      7093325.00
      2784275.04      7093974.98
#Sta/Elev= 30
  3334.3  590.64  4287.7  570.89  4544.0  569.17  4564.5  568.19  4578.8  564.83
  4605.5  561.71  4636.3  561.23  4667.1  562.47  4672.9  567.44  4708.1  563.67
  4808.3  562.44  4926.1  563.88  4932.7  562.01  4938.1  563.78  4962.2  562.15
  4967.6  563.99  4986.2  561.24  4991.6  563.45  4995.7  559.49  4996.2  558.69
  5002.1  559.49  5009.7  564.13  5073.2  563.63  5173.8  564.83  5290.3  567.35
  5526.7  565.69  5711.9  566.87  5937.9  572.71  6358.9  577.47  6650.3  583.49
#Mann=7,-1,0
  3334.3    0.05       0  4808.3    0.12       0  4995.7    0.07       0
  5002.1    0.12       0  5073.2    0.05       0  5526.7    0.16       0
  5937.9    0.05       0
Bank Sta=4578.8,5173.8
Exp/Cntr=0.3,0.1

Type RM Length L Ch R = 1,48045,174,174,174
BEGIN DESCRIPTION:
Mapping XS 360afa89
END DESCRIPTION:
XS GIS Cut Line= 3
      2786478.76      7093105.95      2785645.43      7093027.83
      2785020.41      7093027.83
#Sta/Elev= 30
  4203.1  571.39  4387.7  569.41  4427.8  568.69  4434.8  567.65  4447.9  567.38
  4458.0  568.30  4488.1  567.96  4585.9  564.89  4728.8  563.29  4789.4  562.83
  4798.5  563.96  4803.5  562.82  4809.5  562.64  4861.4  562.28  5000.3  562.05
  5010.4  561.09  5012.8  557.46  5013.3  556.66  5019.0  556.66  5019.5  557.46
  5030.1  558.17  5037.8  561.40  5042.8  561.40  5050.5  563.64  5080.5  562.83
  5258.1  563.15  5269.0  563.29  5520.5  566.38  5600.5  569.85  5665.1  569.89
#Mann=7,-1,0
  4203.1    0.05       0  4434.8    0.08       0  4861.4    0.05       0
  5012.8    0.04       0  5019.5    0.05       0  5030.1    0.12       0
  5258.1    0.08       0
Bank Sta=4728.8,5269
Exp/Cntr=0.3,0.1

Type RM Length L Ch R = 1,47871,540,540,540
BEGIN DESCRIPTION:
CEDAR CREEK 53.0
END DESCRIPTION:
XS GIS Cut Line= 3
      2786457.96      7092913.25      2785625.00      7092875.00
      2784825.04      7092875.00
#Sta/Elev= 30
  4169.0  568.96  4312.1  567.25  4342.1  565.75  4532.3  564.46  4615.7  562.86
  4812.6  561.74  4895.8  562.02  4912.7  563.04  4932.8  559.13  4942.8  561.53
  4952.8  562.44  4982.8  562.44  4992.8  558.63  4997.0  556.02  4997.5  555.22
  5003.2  555.22  5003.7  556.02  5005.3  556.02  5012.8  561.58  5022.8  562.32
  5152.8  561.69  5182.8  560.55  5212.8  561.08  5242.8  559.53  5272.8  562.87
  5308.4  562.86  5332.8  564.01  5402.8  564.15  5632.8  569.39  5802.8  574.31
#Mann=3,-1,0
  4169.0    0.05       0  4997.0    0.04       0  5003.7    0.05       0
Bank Sta=4615.7,5308.4
Exp/Cntr=0.3,0.1

Type RM Length L Ch R = 1,47331,601,601,601
BEGIN DESCRIPTION:
CEDAR CREEK 52.0
END DESCRIPTION:
XS GIS Cut Line= 3
      2786452.75      7092418.45      2785675.00      7092375.00
      2784775.65      7092397.62
#Sta/Elev= 30
  4175.9  569.94  4213.7  569.91  4253.8  568.91  4394.0  568.40  4414.0  569.41
  4434.1  568.33  4624.4  567.01  4682.7  563.65  4764.6  562.18  4778.5  561.36
  4814.6  559.57  4862.5  558.19  4885.3  559.97  4974.9  560.91  4984.9  559.12
  4991.5  555.02  4992.0  554.22  4997.7  554.22  4998.2  555.02  5014.9  560.40
  5024.9  560.99  5126.8  560.87  5245.0  559.76  5398.5  561.36  5475.0  562.35
  5550.8  565.32  5625.1  566.48  5665.1  568.30  5755.1  570.88  5854.5  571.98
#Mann=5,-1,0
  4175.9    0.05       0  4885.3    0.16       0  4991.5    0.07       0
  4998.2    0.16       0  5126.8    0.05       0
Bank Sta=4778.5,5398.5
Exp/Cntr=0.3,0.1

Type RM Length L Ch R = 1,46730,889,889,889
BEGIN DESCRIPTION:
CEDAR CREEK 51.0
END DESCRIPTION:
XS GIS Cut Line= 3
      2786124.98      7092174.99      2785675.00      7091925.00
      2784874.96      7091925.00
#Sta/Elev= 30
  4483.7  567.45  4572.9  566.83  4586.6  567.77  4616.4  566.39  4675.9  565.53
  4800.6  564.95  4918.4  561.25  4936.8  559.97  4944.2  559.69  4968.7  558.01
  4975.6  558.67  4990.4  555.34  4992.2  552.95  4992.7  552.15  4998.5  552.15
  4999.0  552.95  5001.0  552.95  5008.5  558.14  5038.5  559.04  5120.9  557.85
  5168.5  557.34  5248.5  558.36  5338.5  558.06  5358.5  557.29  5438.5  558.98
  5508.5  559.00  5515.8  559.69  5608.5  561.55  5738.5  568.57  5798.5  570.64
#Mann=5,-1,0
  4483.7    0.05       0  4936.8    0.16       0  4992.2    0.07       0
  4999.0    0.16       0  5120.9    0.05       0
Bank Sta=4944.2,5515.8
Exp/Cntr=0.3,0.1

Type RM Length L Ch R = 1,45841,796,796,796
BEGIN DESCRIPTION:
CEDAR CREEK 50.0
END DESCRIPTION:
XS GIS Cut Line= 3
      2785900.62      7091501.78      2785353.76      7091283.04
      2784864.13      7091309.08
#Sta/Elev= 30
  4404.3  565.35  4423.0  565.65  4460.9  563.71  4490.5  563.72  4550.4  560.55
  4574.0  560.76  4615.0  558.18  4650.4  557.68  4676.3  556.27  4722.7  556.21
  4765.0  554.63  4808.2  556.39  4813.6  554.98  4837.8  556.13  4870.7  554.91
  4905.8  554.80  4950.9  556.71  4976.4  556.08  4981.2  555.94  4989.9  551.58
  4998.6  550.24  4999.1  549.44  5005.0  549.44  5005.5  550.24  5012.1  555.29
  5022.1  556.36  5076.8  556.85  5114.0  557.68  5242.4  559.30  5483.6  565.43
#Mann=8,-1,0
  4404.3    0.05       0  4423.0    0.16       0  4765.0    0.05       0
  4870.7    0.12       0  4976.4    0.16       0  4998.6    0.07       0
  5005.5    0.16       0  5076.8    0.05       0
Bank Sta=4650.4,5114
Exp/Cntr=0.3,0.1

Type RM Length L Ch R = 1,45045,565,565,565
BEGIN DESCRIPTION:
CEDAR CREEK 49.0
END DESCRIPTION:
XS GIS Cut Line= 3
      2786009.97      7091022.60      2785325.00      7090625.00
      2784874.97      7090675.00
#Sta/Elev= 30
  4184.7  560.25  4267.6  560.34  4448.5  555.22  4595.1  554.01  4761.6  554.72
  4808.2  554.63  4824.0  552.36  4829.7  554.07  4845.5  553.10  4851.3  554.12
  4895.8  553.94  4910.0  553.55  4931.6  550.82  4941.5  552.87  4947.3  551.16
  4953.6  553.11  4963.1  553.14  4968.8  550.21  4970.2  547.15  4970.8  546.35
  4977.4  547.15  5006.9  548.95  5016.0  552.69  5027.0  551.96  5032.4  555.22
  5037.1  558.06  5047.1  558.88  5077.3  558.44  5167.9  561.91  5429.5  568.65
#Mann=5,-1,0
  4184.7    0.05       0  4761.6    0.16       0  4970.2    0.07       0
  4977.4    0.16       0  5016.0    0.05       0
Bank Sta=4448.5,5032.4
Exp/Cntr=0.3,0.1

Type RM Length L Ch R = 1,44480,822,822,822
BEGIN DESCRIPTION:
CEDAR CREEK 48.0
END DESCRIPTION:
XS GIS Cut Line= 3
      2787125.03      7091175.02      2785575.00      7090225.00
      2785025.00      7089925.00
#Sta/Elev= 30
  3218.2  570.91  3800.4  559.96  4121.4  561.46  4373.7  554.08  4648.7  551.67
  4672.1  552.31  4759.7  550.91  4833.1  553.30  4906.6  551.50  4970.5  552.41
  4985.9  550.74  4991.8  545.76  4997.4  545.65  4997.9  544.85  5004.7  545.65
  5007.2  545.96  5013.1  552.59  5022.6  553.26  5100.1  554.08  5173.3  557.38
  5300.6  561.22  5322.4  558.06  5338.5  560.95  5382.2  562.23  5404.0  560.77
  5442.0  562.89  5463.8  560.78  5491.8  564.31  5545.5  566.79  5662.7  569.34
#Mann=7,-1,0
  3218.2    0.05       0  4648.7    0.16       0  4672.1    0.12       0
  4997.4    0.07       0  5004.7    0.12       0  5022.6    0.16       0
  5173.3    0.05       0
Bank Sta=4373.7,5100.1
Exp/Cntr=0.3,0.1

Type RM Length L Ch R = 1,43658,822,822,822
BEGIN DESCRIPTION:
CEDAR CREEK 47.0
END DESCRIPTION:
XS GIS Cut Line= 3
      2786724.99      7089998.61      2786275.00      7089948.61
      2785624.98      7089898.61
#Sta/Elev= 30
  4539.9  558.59  4640.5  557.19  4700.9  558.16  4841.7  552.68  4883.9  552.16
  4952.4  551.52  4974.9  550.06  4978.8  549.99  4983.9  548.60  4986.4  544.67
  4987.0  543.87  4993.3  543.87  4993.8  544.67  5012.7  550.97  5101.5  550.78
  5123.0  549.70  5163.2  549.48  5193.3  550.70  5253.4  549.64  5273.5  550.11
  5283.5  547.46  5311.2  550.53  5372.6  552.16  5434.0  553.06  5454.0  554.17
  5497.6  554.45  5594.4  557.25  5614.5  558.99  5623.0  558.27  5644.6  558.55
#Mann=5,-1,0
  4539.9    0.05       0  4974.9    0.12       0  4986.4    0.07       0
  4993.8    0.12       0  5311.2    0.16       0
Bank Sta=4883.9,5372.6
Exp/Cntr=0.3,0.1

Type RM Length L Ch R = 1,42836,107,107,107
BEGIN DESCRIPTION:
CEDAR CREEK 46.0
END DESCRIPTION:
XS GIS Cut Line= 3
      2786674.97      7089674.98      2786175.00      7089325.00
      2785725.04      7089125.02
#Sta/Elev= 30
  4375.3  558.13  4525.7  552.38  4635.4  550.25  4923.0  547.87  4942.4  546.63
  4949.0  544.82  4963.4  544.13  4972.1  541.94  4978.2  543.91  4982.5  541.52
  4990.7  540.92  4991.3  540.12  4997.7  540.12  4998.3  540.92  5000.0  541.05
  5007.5  545.14  5023.2  548.27  5040.3  548.02  5046.5  547.18  5051.9  545.04
  5069.7  548.22  5098.4  547.93  5147.0  550.25  5220.2  552.71  5271.3  555.76
  5281.1  555.43  5302.9  556.73  5388.4  557.75  5440.4  558.45  5478.0  560.09
#Mann=6,-1,0
  4375.3    0.05       0  4923.0    0.16       0  4990.7    0.07       0
  4998.3    0.16       0  5271.3    0.05       0  5388.4    0.16       0
Bank Sta=4635.4,5147
Exp/Cntr=0.3,0.1

Type RM Length L Ch R = 1,42729,204,204,204
BEGIN DESCRIPTION:
Mapping XS ae664961
END DESCRIPTION:
XS GIS Cut Line= 3
      2787011.13      7089240.50      2786143.12      7089227.48
      2785761.14      7089092.92
#Sta/Elev= 30
  4115.1  556.94  4211.2  556.89  4281.3  554.58  4331.3  554.68  4351.3  555.76
  4401.3  554.57  4431.3  552.85  4679.1  549.15  4816.6  548.61  4851.3  548.63
  4881.3  547.44  4915.7  548.32  4983.2  548.02  4991.8  545.06  4997.6  540.15
  4998.2  539.35  5004.6  539.35  5005.2  540.15  5006.7  540.18  5013.0  545.30
  5016.4  546.14  5023.6  547.91  5037.7  546.82  5061.7  549.15  5170.8  552.19
  5224.7  555.03  5243.7  555.37  5280.0  558.02  5331.1  559.13  5388.2  558.07
#Mann=8,-1,0
  4115.1    0.05       0  4816.6    0.16       0  4915.7    0.05       0
  4997.6    0.03       0  5005.2    0.05       0  5016.4    0.16       0
  5170.8    0.08       0  5224.7    0.16       0
Bank Sta=4679.1,5061.7
Exp/Cntr=0.3,0.1

Type RM Length L Ch R = 1,42525,292,292,292
BEGIN DESCRIPTION:
Mapping XS d8f68ab7
END DESCRIPTION:
XS GIS Cut Line= 4
      2787028.55      7089075.57      2786125.75      7089019.15
      2785939.12      7088997.45      2785713.45      7088893.29
#Sta/Elev= 30
  4090.4  557.89  4214.2  555.06  4284.3  555.42  4544.8  548.63  4735.2  546.59
  4890.5  547.38  4915.6  547.06  4925.6  544.54  4935.6  544.52  4945.6  546.74
  4975.7  547.54  4986.0  546.89  4992.8  543.72  4997.9  543.72  5002.0  541.52
  5002.6  540.72  5009.6  541.52  5025.9  547.31  5103.7  547.58  5126.6  547.42
  5142.3  548.63  5166.9  554.87  5219.7  556.06  5254.7  555.39  5271.1  555.73
  5276.6  554.52  5312.8  553.86  5317.0  553.73  5322.5  555.99  5431.4  557.46
#Mann=7,-1,0
  4090.4    0.05       0  4890.5    0.12       0  5002.0    0.07       0
  5009.6    0.12       0  5103.7    0.05       0  5254.7    0.16       0
  5312.8    0.05       0
Bank Sta=4544.8,5142.3
Exp/Cntr=0.3,0.1

Type RM Length L Ch R = 1,42233,532,532,532
BEGIN DESCRIPTION:
Mapping XS 21bed44d
END DESCRIPTION:
XS GIS Cut Line= 3
      2786998.13      7088793.45      2786190.86      7088763.07
      2785761.15      7088815.16
#Sta/Elev= 30
  4185.8  556.01  4219.0  556.20  4269.0  554.08  4369.1  552.80  4517.3  548.12
  4579.2  546.70  4599.2  547.15  4619.2  545.82  4719.3  546.09  4734.1  544.52
  4759.3  541.82  4779.4  544.35  4799.4  544.81  4819.4  546.94  4889.4  546.35
  4979.5  547.11  4993.6  545.97  4995.7  539.19  4996.3  538.39  5002.7  538.39
  5003.3  539.19  5009.6  545.02  5019.7  546.82  5029.8  545.76  5047.3  548.12
  5080.1  549.63  5160.7  550.47  5220.9  552.47  5362.9  555.68  5426.5  556.90
#Mann=6,-1,0
  4185.8    0.05       0  4734.1    0.12       0  4995.7    0.07       0
  5003.3    0.12       0  5220.9    0.16       0  5362.9    0.05       0
Bank Sta=4517.3,5047.3
Exp/Cntr=0.3,0.1

Type RM Length L Ch R = 1,41701,233,233,233
BEGIN DESCRIPTION:
Mapping XS 02f6d5fb
END DESCRIPTION:
XS GIS Cut Line= 3
      2786959.04      7088533.03      2786360.13      7088502.65
      2785821.96      7088559.08
#Sta/Elev= 30
  4388.3  555.27  4432.4  553.97  4492.5  553.37  4542.5  550.52  4582.6  549.65
  4612.6  547.53  4633.1  547.28  4662.7  546.16  4682.7  546.58  4702.7  545.20
  4782.8  545.73  4792.9  543.27  4802.9  539.92  4814.4  544.31  4822.9  546.19
  4883.0  545.51  4988.0  545.53  4993.1  544.71  5003.2  540.31  5009.4  539.41
  5010.0  538.61  5016.4  538.61  5017.0  539.41  5023.3  546.08  5063.5  545.30
  5216.2  547.28  5348.1  550.53  5375.2  552.54  5490.1  554.51  5529.1  554.82
#Mann=5,-1,0
  4388.3    0.05       0  4814.4    0.12       0  5009.4    0.07       0
  5017.0    0.12       0  5490.1    0.16       0
Bank Sta=4633.1,5216.2
Exp/Cntr=0.3,0.1

Type RM Length L Ch R = 1,41468,743,743,743
BEGIN DESCRIPTION:
CEDAR CREEK 43.0
END DESCRIPTION:
XS GIS Cut Line= 3
      2786937.41      7088398.49      2786342.77      7088333.38
      2785749.07      7088116.70
#Sta/Elev= 30
  4332.3  553.87  4385.0  553.85  4529.6  546.89  4636.5  544.40  4692.3  545.47
  4717.0  544.95  4727.1  539.16  4747.2  545.60  4857.8  545.23  4871.3  544.16
  4972.8  545.00  4981.3  543.43  4992.0  539.97  4994.2  537.73  4994.8  536.93
  5001.3  536.93  5001.9  537.73  5003.3  541.45  5013.3  544.99  5045.2  544.59
  5084.3  546.42  5176.6  546.25  5214.4  546.89  5240.9  547.25  5292.9  549.29
  5298.4  548.18  5300.7  547.72  5318.1  549.69  5435.0  550.62  5562.5  553.26
#Mann=7,-1,0
  4332.3    0.05       0  4692.3    0.12       0  4994.2    0.07       0
  5001.9    0.12       0  5176.6    0.16       0  5240.9    0.12       0
  5298.4    0.16       0
Bank Sta=4529.6,5214.4
Exp/Cntr=0.3,0.1

Type RM Length L Ch R = 1,40725,673,673,673
BEGIN DESCRIPTION:
CEDAR CREEK 42.0
END DESCRIPTION:
XS GIS Cut Line= 3
      2787122.58      7087922.19      2786487.69      7087913.08
      2785628.55      7087965.71
#Sta/Elev= 30
  4293.8  552.71  4341.4  552.11  4381.4  552.93  4481.4  550.42  4561.4  551.15
  4631.4  548.91  4691.4  550.49  4822.6  545.60  4838.0  545.37  4871.4  544.02
  4881.4  542.95  4891.4  540.35  4901.4  539.71  4911.4  542.36  4921.4  543.50
  4981.5  543.47  4991.6  541.82  4997.6  535.65  4998.3  534.85  5004.9  534.85
  5005.5  535.65  5011.6  536.60  5021.6  543.40  5031.6  544.21  5275.0  543.60
  5446.6  545.60  5492.5  546.33  5662.8  553.84  5722.9  554.36  5789.5  558.07
#Mann=5,-1,0
  4293.8    0.05       0  4838.0    0.12       0  4997.6    0.07       0
  5005.5    0.12       0  5275.0    0.05       0
Bank Sta=4822.6,5446.6
Exp/Cntr=0.3,0.1

Type RM Length L Ch R = 1,40052,638,638,638
BEGIN DESCRIPTION:
CEDAR CREEK 41.0
END DESCRIPTION:
XS GIS Cut Line= 3
      2787084.92      7087660.63      2786468.64      7087500.05
      2785709.57      7087426.31
#Sta/Elev= 30
  4158.4  550.51  4189.3  550.74  4261.7  548.87  4292.7  549.41  4400.0  548.50
  4435.3  546.72  4481.0  546.35  4514.5  544.54  4644.0  542.36  4654.3  540.90
  4673.2  542.76  4712.6  542.26  4794.6  543.22  4901.8  541.91  4979.8  542.34
  4989.8  541.23  4999.8  534.77  5000.5  533.97  5007.1  533.97  5007.7  534.77
  5009.9  537.45  5020.0  542.93  5057.8  542.59  5225.2  544.54  5308.7  546.63
  5371.6  548.02  5381.6  548.44  5391.7  550.51  5518.5  554.49  5557.9  556.52
#Mann=6,-1,0
  4158.4    0.05       0  4712.6    0.12       0  4999.8    0.07       0
  5007.7    0.12       0  5057.8    0.16       0  5308.7    0.05       0
Bank Sta=4514.5,5225.2
Exp/Cntr=0.3,0.1

Type RM Length L Ch R = 1,39414,591,591,591
BEGIN DESCRIPTION:
CEDAR CREEK 40.0
END DESCRIPTION:
XS GIS Cut Line= 3
      2787109.23      7087355.07      2786718.64      7087209.25
      2785808.63      7087235.25
#Sta/Elev= 30
  4575.5  548.42  4819.5  545.75  4844.4  546.41  4857.5  545.37  4905.0  545.54
  4954.3  544.44  4975.0  544.04  4976.9  542.99  4985.3  538.40  4990.6  538.84
  4996.7  537.67  5002.1  534.24  5002.8  533.44  5009.4  533.44  5010.1  534.24
  5014.9  535.79  5019.9  539.66  5026.1  541.19  5041.2  541.33  5146.1  541.65
  5236.2  539.87  5266.2  541.65  5316.2  541.17  5386.2  542.38  5455.8  542.45
  5498.8  542.99  5626.3  544.43  5713.4  546.40  5786.4  550.08  5902.8  552.53
#Mann=7,-1,0
  4575.5    0.05       0  4954.3    0.16       0  5002.1    0.07       0
  5010.1    0.16       0  5041.2    0.12       0  5455.8    0.16       0
  5713.4    0.05       0
Bank Sta=4976.9,5498.8
Exp/Cntr=0.3,0.1

Type RM Length L Ch R = 1,38823,608,608,608
BEGIN DESCRIPTION:
CEDAR CREEK 39.0
END DESCRIPTION:
XS GIS Cut Line= 3
      2787213.39      7087297.76      2786645.72      7086782.17
      2786104.80      7086589.73
#Sta/Elev= 30
  4240.2  547.05  4593.3  541.84  4737.9  539.60  4828.7  539.96  4842.9  536.64
  4852.1  535.89  4857.1  536.05  4871.3  540.00  4906.5  539.57  4913.5  538.83
  4920.6  536.17  4934.8  539.57  4963.2  540.29  4970.0  540.08  4977.4  535.36
  4980.1  532.10  4980.8  531.30  4988.2  532.10  4991.6  534.51  4998.4  534.05
  5004.2  537.52  5010.1  537.52  5013.3  539.36  5018.6  533.02  5029.1  539.32
  5038.9  539.99  5162.4  541.84  5316.7  546.35  5386.9  548.37  5581.2  554.37
#Mann=7,-1,0
  4240.2    0.05       0  4737.9    0.16       0  4852.1    0.12       0
  4980.1    0.07       0  4988.2    0.12       0  5316.7    0.16       0
  5386.9    0.05       0
Bank Sta=4593.3,5162.4
Exp/Cntr=0.3,0.1

Type RM Length L Ch R = 1,38215,628,628,628
BEGIN DESCRIPTION:
Mapping XS 67cfbca5
END DESCRIPTION:
XS GIS Cut Line= 3
      2787270.73      7087276.99      2786958.22      7086641.54
      2786560.08      7086289.94
#Sta/Elev= 30
  4271.3  546.05  4306.9  545.39  4337.9  543.13  4463.0  543.64  4603.2  540.75
  4644.1  540.38  4750.1  539.76  4815.4  538.95  4910.9  539.68  4942.1  538.77
  4955.8  536.02  4972.7  536.32  4975.0  535.48  4979.4  534.60  4986.1  530.67
  4989.6  530.32  4990.3  529.52  4997.7  530.32  5000.3  532.27  5007.9  533.41
  5014.5  537.76  5028.8  538.78  5128.3  539.44  5170.5  539.11  5177.7  537.85
  5184.3  539.09  5318.8  540.75  5334.1  540.75  5418.6  544.51  5510.6  546.74
#Mann=7,-1,0
  4271.3    0.05       0  4644.1    0.12       0  4750.1    0.16       0
  4975.0    0.12       0  4989.6    0.07       0  4997.7    0.12       0
  5318.8    0.16       0
Bank Sta=4603.2,5334.1
Exp/Cntr=0.3,0.1

Type RM Length L Ch R = 1,37587,389,389,389
BEGIN DESCRIPTION:
double CEDAR CREEK 38.0
END DESCRIPTION:
XS GIS Cut Line= 3
      2787575.02      7086775.01      2787165.57      7086381.88
      2786725.03      7086075.02
#Sta/Elev= 30
  4432.8  545.39  4454.0  545.37  4517.6  543.00  4753.6  538.81  4814.8  536.18
  4821.7  534.70  4828.9  536.43  4860.8  536.97  4892.6  537.41  4963.2  537.89
  4977.3  536.92  4984.6  533.97  4991.5  532.49  4993.2  528.29  4993.9  527.49
  5000.9  527.49  5001.6  528.29  5005.5  529.08  5013.3  537.05  5020.3  538.54
  5157.3  537.29  5243.7  537.54  5266.3  538.81  5318.4  539.87  5351.0  540.92
  5372.0  540.28  5422.6  542.75  5443.5  542.81  5509.7  545.30  5537.3  545.71
#Mann=7,-1,0
  4432.8    0.05       0  4860.8    0.16       0  4892.6    0.12       0
  4993.2    0.07       0  5001.6    0.12       0  5318.4    0.16       0
  5509.7    0.05       0
Bank Sta=4753.6,5266.3
Exp/Cntr=0.3,0.1

Type RM Length L Ch R = 1,37198,686,686,686
BEGIN DESCRIPTION:
double CEDAR CREEK 37.0
END DESCRIPTION:
XS GIS Cut Line= 3
      2788072.76      7086552.97      2787325.00      7086075.00
      2786525.00      7085675.00
#Sta/Elev= 30
  4150.9  544.30  4577.3  538.20  4761.2  535.69  4812.9  534.94  4967.2  536.77
  4973.2  535.42  4979.2  536.51  4988.5  531.01  4994.4  534.68  4998.5  528.03
  4999.3  527.23  5007.0  528.03  5009.6  533.92  5015.5  528.53  5024.8  535.05
  5046.8  536.62  5262.0  536.08  5270.4  532.49  5276.0  532.40  5292.7  535.96
  5337.4  536.88  5343.0  535.38  5351.4  535.69  5387.8  540.27  5449.2  540.62
  5454.8  539.08  5482.6  538.20  5530.6  541.71  5701.0  546.90  5932.8  553.72
#Mann=6,-1,0
  4150.9    0.05       0  4761.2    0.12       0  4998.5    0.07       0
  5007.0    0.12       0  5530.6    0.16       0  5701.0    0.05       0
Bank Sta=4577.3,5482.6
Exp/Cntr=0.3,0.1

Type RM Length L Ch R = 1,36512,573,573,573
BEGIN DESCRIPTION:
CEDAR CREEK 36.0
END DESCRIPTION:
XS GIS Cut Line= 3
      2788474.97      7086424.97      2787725.00      7085675.00
      2786875.03      7085275.01
#Sta/Elev= 30
  3921.5  548.80  4133.6  545.35  4402.3  538.41  4584.1  537.09  4768.5  535.16
  4825.3  535.06  4897.3  534.45  4911.4  531.66  4925.5  534.35  4968.0  534.77
  4984.9  533.22  4990.8  525.62  4992.0  525.38  4992.8  524.58  5000.6  525.38
  5004.2  529.09  5013.5  534.27  5103.7  534.84  5161.4  536.56  5170.0  536.31
  5178.6  532.32  5184.2  536.45  5201.4  535.65  5207.0  537.12  5217.7  537.09
  5236.3  538.27  5280.9  537.59  5460.8  540.07  5719.5  546.56  5921.5  548.92
#Mann=6,-1,0
  3921.5    0.05       0  4768.5    0.16       0  4825.3    0.12       0
  4992.0    0.07       0  5000.6    0.12       0  5460.8    0.05       0
Bank Sta=4584.1,5217.7
Exp/Cntr=0.3,0.1

Type RM Length L Ch R = 1,35939,398,398,398
BEGIN DESCRIPTION:
CEDAR CREEK 35.0
END DESCRIPTION:
XS GIS Cut Line= 3
      2788437.35      7085417.57      2788025.00      7085275.00
      2786725.04      7085175.00
#Sta/Elev= 30
  4538.7  544.97  4583.5  545.17  4699.9  542.36  4741.2  542.19  4784.5  538.46
  4816.3  538.66  4901.7  534.48  4909.7  534.28  4977.5  533.74  4982.0  531.42
  4985.0  529.87  4990.7  524.51  4991.5  523.71  4998.6  523.71  4999.4  524.51
  5005.1  528.56  5015.1  533.53  5045.2  533.25  5065.3  534.16  5095.4  531.38
  5145.5  533.58  5195.7  532.56  5225.7  533.33  5235.8  532.67  5265.9  534.14
  5410.8  534.48  5626.9  536.60  5698.1  539.08  5947.9  546.14  6278.8  551.12
#Mann=6,-1,0
  4538.7    0.16       0  4909.7    0.05       0  4982.0    0.12       0
  4990.7    0.07       0  4999.4    0.12       0  5698.1    0.05       0
Bank Sta=4901.7,5410.8
Exp/Cntr=0.3,0.1

Type RM Length L Ch R = 1,35541,717,717,717
BEGIN DESCRIPTION:
CEDAR CREEK 34.0
END DESCRIPTION:
XS GIS Cut Line= 3
      2788489.48      7085172.80      2788031.14      7084907.17
      2787048.36      7084730.37
#Sta/Elev= 30
  4457.8  543.92  4511.5  543.13  4621.0  542.70  4626.7  541.36  4765.9  539.07
  4824.7  536.55  4860.4  533.23  4963.9  531.13  4971.5  531.87  4979.6  530.25
  4984.7  526.30  4999.6  523.90  5000.3  523.10  5008.3  523.90  5013.3  524.53
  5023.6  528.72  5027.3  531.45  5028.7  532.48  5034.4  532.57  5199.8  532.75
  5278.3  531.18  5484.9  533.23  5517.6  533.67  5603.9  535.94  5623.7  536.42
  5727.8  539.02  5755.8  539.38  5766.7  537.92  5849.7  541.68  5986.1  545.26
#Mann=11,-1,0
  4457.8    0.16       0  4511.5    0.05       0  4999.6    0.03       0
  5008.3    0.05       0  5013.3    0.16       0  5027.3    0.12       0
  5517.6    0.05       0  5603.9    0.16       0  5623.7    0.12       0
  5727.8    0.16       0  5849.7    0.05       0
Bank Sta=4860.4,5484.9
Exp/Cntr=0.3,0.1

Type RM Length L Ch R = 1,34824,549,549,549
BEGIN DESCRIPTION:
CEDAR CREEK 33.0
END DESCRIPTION:
XS GIS Cut Line= 3
      2788827.99      7084657.16      2788175.00      7084425.00
      2787573.26      7084219.82
#Sta/Elev= 30
  4280.5  542.31  4449.7  539.38  4517.2  539.44  4612.7  535.41  4629.4  536.60
  4634.7  535.45  4655.0  535.56  4743.8  532.08  4771.9  530.97  4901.7  530.08
  4967.0  531.03  4983.9  531.23  4989.2  529.36  4994.7  525.33  5000.8  523.60
  5001.6  522.80  5009.7  523.60  5015.3  531.15  5020.5  531.32  5114.6  529.48
  5217.3  530.10  5227.1  528.38  5248.2  529.92  5356.0  529.77  5396.8  532.08
  5459.8  535.38  5480.1  535.66  5516.7  538.85  5574.1  537.73  5609.3  538.63
#Mann=7,-1,0
  4280.5    0.05       0  4967.0    0.16       0  5000.8    0.07       0
  5009.7    0.16       0  5217.3    0.12       0  5356.0    0.16       0
  5459.8    0.05       0
Bank Sta=4743.8,5396.8
Exp/Cntr=0.3,0.1

Type RM Length L Ch R = 1,34275,557,557,557
BEGIN DESCRIPTION:
CEDAR CREEK 32.0
END DESCRIPTION:
XS GIS Cut Line= 3
      2788874.96      7084124.99      2788425.00      7083975.00
      2787688.66      7084016.47
#Sta/Elev= 30
  4523.2  540.98  4565.3  539.39  4607.5  537.03  4691.8  535.23  4734.0  532.78
  4786.7  531.93  4818.0  530.59  4892.1  528.34  4904.2  527.22  4934.3  529.30
  4965.9  529.73  4987.0  529.21  4994.9  527.96  5000.0  527.96  5003.0  521.96
  5003.9  521.16  5011.2  521.16  5012.0  521.96  5027.5  528.71  5037.6  529.76
  5077.6  529.87  5107.7  529.11  5207.8  529.74  5237.9  529.36  5257.9  528.42
  5268.6  529.22  5447.0  530.59  5518.3  532.46  5621.7  538.57  5735.0  539.37
#Mann=4,-1,0
  4523.2    0.05       0  4904.2    0.07       0  5003.0    0.07       0
  5012.0    0.05       0
Bank Sta=4818,5447
Exp/Cntr=0.3,0.1

Type RM Length L Ch R = 1,33718,756,756,756
BEGIN DESCRIPTION:
CEDAR CREEK 31.0
END DESCRIPTION:
XS GIS Cut Line= 3
      2789074.97      7083924.98      2788619.68      7083620.71
      2787839.23      7083657.13
#Sta/Elev= 30
  4463.8  544.14  4477.3  542.64  4564.4  539.77  4657.5  537.92  4723.5  535.64
  4744.6  536.23  4765.6  535.79  4824.6  533.25  4873.7  532.86  4903.7  530.94
  4924.8  530.51  4932.4  529.40  4960.8  528.64  4981.8  526.35  4986.3  525.21
  4987.2  524.41  4994.5  524.41  4995.3  525.21  5005.0  528.05  5011.2  528.71
  5306.4  528.18  5326.4  525.92  5346.4  528.44  5366.5  527.57  5456.6  527.05
  5621.2  529.40  5696.8  530.66  5756.9  532.89  5776.9  532.93  5792.7  531.96
#Mann=3,-1,0
  4463.8    0.05       0  4986.3    0.03       0  4995.3    0.05       0
Bank Sta=4932.4,5621.2
Exp/Cntr=0.3,0.1

Type RM Length L Ch R = 1,32962,561,561,561
BEGIN DESCRIPTION:
CEDAR CREEK 30.0
END DESCRIPTION:
XS GIS Cut Line= 3
      2788925.03      7083325.01      2788325.00      7083225.00
      2787725.02      7082925.01
#Sta/Elev= 30
  4380.5  535.06  4421.1  533.95  4492.0  533.70  4552.9  531.04  4583.3  531.76
  4644.1  530.76  4717.6  531.04  4745.5  528.07  4791.5  527.45  4857.0  526.21
  4968.5  526.86  4978.7  524.29  4981.8  519.94  4982.6  519.14  4990.0  519.14
  4990.8  519.94  4997.2  522.12  5002.8  520.69  5011.2  526.08  5019.6  526.81
  5198.1  526.36  5271.1  526.41  5293.5  525.35  5301.9  522.65  5307.6  524.37
  5310.2  525.16  5332.6  525.79  5379.2  525.86  5419.3  527.45  5659.6  537.25
#Mann=6,-1,0
  4380.5    0.05       0  4981.8    0.03       0  4990.8    0.05       0
  5198.1    0.16       0  5307.6    0.12       0  5379.2    0.16       0
Bank Sta=4791.5,5419.3
Exp/Cntr=0.3,0.1

Type RM Length L Ch R = 1,32401,616,616,616
BEGIN DESCRIPTION:
CEDAR CREEK 29.0
END DESCRIPTION:
XS GIS Cut Line= 3
      2789174.98      7082925.00      2788225.00      7082725.00
      2787775.00      7082725.00
#Sta/Elev= 30
  4018.8  540.40  4029.0  537.78  4049.4  535.29  4069.9  534.41  4172.1  533.69
  4366.2  530.33  4476.7  529.87  4618.2  526.09  4764.8  525.05  4795.4  523.62
  4836.3  525.07  4897.6  524.42  4967.8  525.58  4979.4  525.78  4987.0  524.08
  4992.1  524.08  4995.0  518.75  4995.9  517.95  5003.4  517.95  5004.3  518.75
  5009.6  518.76  5019.6  525.21  5129.6  523.90  5149.6  525.39  5159.6  524.55
  5209.6  524.92  5227.6  526.09  5279.6  532.16  5343.2  535.91  5439.6  538.73
#Mann=5,-1,0
  4018.8    0.05       0  4967.8    0.12       0  4995.0    0.07       0
  5004.3    0.12       0  5343.2    0.05       0
Bank Sta=4618.2,5227.6
Exp/Cntr=0.3,0.1

Type RM Length L Ch R = 1,31785,286,286,286
BEGIN DESCRIPTION:
Mapping XS b0ed2c10
END DESCRIPTION:
XS GIS Cut Line= 6
      2789156.10      7082334.25      2788812.39      7082282.17
      2788676.97      7082193.63      2788057.18      7082172.79
      2787911.34      7082172.79      2787703.74      7082240.26
#Sta/Elev= 30
  3872.5  530.01  3974.8  529.78  4169.9  526.67  4244.6  527.24  4280.8  526.48
  4288.7  525.36  4320.6  524.95  4494.4  523.12  4604.0  523.59  4634.0  521.39
  4644.1  521.36  4674.1  523.24  4783.3  523.14  4799.8  524.24  4874.2  523.21
  4974.2  524.07  4994.3  517.69  4996.0  515.57  4996.9  514.77  5004.4  514.77
  5005.3  515.57  5014.3  518.75  5024.3  523.50  5034.3  524.28  5097.3  524.57
  5127.9  524.95  5234.7  527.24  5335.8  531.28  5355.7  531.30  5366.2  531.57
#Mann=6,-1,0
  3872.5    0.05       0  4799.8    0.12       0  4996.0    0.07       0
  5005.3    0.12       0  5097.3    0.05       0  5355.7    0.16       0
Bank Sta=4320.6,5127.9
Exp/Cntr=0.3,0.1

Type RM Length L Ch R = 1,31499,506,506,506
BEGIN DESCRIPTION:
Mapping XS 8b6594df
END DESCRIPTION:
XS GIS Cut Line= 5
      2789286.33      7082178.00      2788817.59      7082110.29
      2788687.39      7082079.04      2788234.26      7082026.96
      2787421.74      7081943.62
#Sta/Elev= 30
  3920.6  530.79  4078.5  528.87  4356.1  526.66  4480.4  525.68  4510.5  524.60
  4668.6  522.55  4852.6  522.40  4873.9  520.10  4882.8  517.99  4892.9  522.15
  4902.9  522.99  4933.1  522.04  4963.3  523.38  4973.4  522.36  4981.3  516.76
  4986.4  516.76  4988.9  515.49  4989.8  514.69  4998.2  515.49  5003.6  516.20
  5013.6  520.74  5023.7  523.30  5291.6  522.83  5375.5  522.97  5414.2  524.60
  5442.7  526.11  5506.2  526.25  5536.4  528.42  5650.9  530.34  5801.0  536.33
#Mann=9,-1,0
  3920.6    0.05       0  4078.5    0.16       0  4356.1    0.08       0
  4480.4    0.05       0  4668.6    0.12       0  4988.9    0.07       0
  4998.2    0.12       0  5291.6    0.16       0  5650.9    0.05       0
Bank Sta=4510.5,5414.2
Exp/Cntr=0.3,0.1

Type RM Length L Ch R = 1,30993,970,970,970
BEGIN DESCRIPTION:
Mapping XS 7882b717
END DESCRIPTION:
XS GIS Cut Line= 3
      2789104.01      7081980.07      2788130.09      7081688.42
      2787541.58      7081657.17
#Sta/Elev= 30
  3980.4  528.73  4132.2  526.70  4282.1  524.75  4303.0  525.41  4355.4  523.84
  4374.4  523.86  4459.6  524.75  4543.0  523.98  4616.1  522.34  4637.0  519.40
  4657.9  521.80  4680.9  521.70  4689.2  521.14  4699.6  515.59  4714.0  520.80
  4720.5  521.99  4767.6  521.17  4971.1  522.01  4981.5  521.56  4989.6  514.67
  4990.5  513.87  4998.9  514.67  5012.2  522.00  5151.6  521.05  5349.8  523.84
  5392.7  526.48  5450.7  528.16  5502.9  529.28  5549.8  531.68  5586.4  532.79
#Mann=9,-1,0
  3980.4    0.05       0  4132.2    0.16       0  4374.4    0.05       0
  4543.0    0.16       0  4767.6    0.12       0  4989.6    0.07       0
  4998.9    0.12       0  5450.7    0.16       0  5549.8    0.05       0
Bank Sta=4355.4,5349.8
Exp/Cntr=0.3,0.1
