--- CHAFFIN CREEK.prj (project) ---

Proj Title=CHAFFIN CREEK Base Level Engineering
Current Plan=p01
Default Exp/Contr=0.3,0.1
English Units
Geom File=g01
Flow File=f01
Plan File=p01
BEGIN DESCRIPTION:
CHAFFIN CREEK
END DESCRIPTION:

--- CHAFFIN CREEK.p01 (plan) ---

Plan Title=Multiple Run
Short Identifier=Multiple
Geom File=g01
Flow File=f01
Subcritical Flow
K Sum by GR= 0
Std Step Tol= 0.01
Critical Tol= 0.01
Num of Std Step Trials= 20
Max Error Tol= 0.3
Flow Tol Ratio= 0.001
Split Flow NTrial= 30
Split Flow Tol= 0.02
Split Flow Ratio= 0.02
Log Output Level= 0
Friction Slope Method= 1
Unsteady Friction Slope Method= 2
Unsteady Bridges Friction Slope Method= 1
Parabolic Critical Depth
Global Vel Dist=  1 , 1 , 1
Global Log Level= 0
CheckData=True
Encroach Param= -1, 0, 0, 0
BEGIN DESCRIPTION:
Multiple Run
END DESCRIPTION:

--- CHAFFIN CREEK.f01 (steady flow) ---

Flow Title=Multiple
Program Version=5.07
Number of Profiles= 7
Profile Names=10-year,25-year,50-year,1pct_min,100-year,1pct_plu,500-year
River Rch & RM=CHAFFIN CREEK,Reach-1         ,27004
     790    1054    1265     753    1502    2997    2112
River Rch & RM=CHAFFIN CREEK,Reach-1         ,23762
     917    1236    1494     895    1786    3563    2545
River Rch & RM=CHAFFIN CREEK,Reach-1         ,22555
    1070    1450    1760    1057    2109    4207    3022
River Rch & RM=CHAFFIN CREEK,Reach-1         ,18684
    1131    1537    1869    1125    2244    4478    3228
River Rch & RM=CHAFFIN CREEK,Reach-1         ,17590
    1314    1804    2210    1339    2671    5329    3895
River Rch & RM=CHAFFIN CREEK,Reach-1         ,16873
    1488    2051    2518    1528    3049    6083    4462
River Rch & RM=CHAFFIN CREEK,Reach-1         ,14183
    1668    2311    2848    1734    3460    6903    5098
River Rch & RM=CHAFFIN CREEK,Reach-1         ,12457
    1706    2366    2918    1778    3547    7077    5233
River Rch & RM=CHAFFIN CREEK,Reach-1         ,11358
    1734    2407    2968    1808    3606    7196    5320
River Rch & RM=CHAFFIN CREEK,Reach-1         ,9017
    2645    3745    4682    2888    5762   11496    8717
River Rch & RM=CHAFFIN CREEK,Reach-1         ,6375
    2821    4007    5019    3102    6189   12348    9398
River Rch & RM=CHAFFIN CREEK,Reach-1         ,4155
    2883    4088    5114    3155    6296   12561    9531
Boundary for River Rch & Prof#=CHAFFIN CREEK,Reach-1         , 1
Up Type= 0
Dn Type= 3
Dn Slope=0.005
Boundary for River Rch & Prof#=CHAFFIN CREEK,Reach-1         , 2
Up Type= 0
Dn Type= 3
Dn Slope=0.005
Boundary for River Rch & Prof#=CHAFFIN CREEK,Reach-1         , 3
Up Type= 0
Dn Type= 3
Dn Slope=0.005
Boundary for River Rch & Prof#=CHAFFIN CREEK,Reach-1         , 4
Up Type= 0
Dn Type= 3
Dn Slope=0.005
Boundary for River Rch & Prof#=CHAFFIN CREEK,Reach-1         , 5
Up Type= 0
Dn Type= 3
Dn Slope=0.005
Boundary for River Rch & Prof#=CHAFFIN CREEK,Reach-1         , 6
Up Type= 0
Dn Type= 3
Dn Slope=0.005
Boundary for River Rch & Prof#=CHAFFIN CREEK,Reach-1         , 7
Up Type= 0
Dn Type= 3
Dn Slope=0.005
DSS Import GetInterval= 0
DSS Import GetPeak= 0
DSS Import FillOption= 0

--- CHAFFIN CREEK.g01 (geometry) ---

Geom Title=Existing Conditions

River Reach=CHAFFIN CREEK,Reach-1
Reach XY= 30
      2831155.59      7089210.71      2831173.72      7088834.41
      2831559.39      7088752.29      2831451.53      7088387.90
      2831942.12      7087909.10      2831767.87      7087561.67
      2832144.61      7087239.74      2832514.56      7086250.46
      2832327.20      7086067.12      2832561.92      7085860.07
      2832172.59      7085577.64      2832835.62      7084430.45
      2833817.93      7083508.58      2834405.82      7083501.23
      2834943.69      7082324.36      2836008.79      7081258.20
      2836511.73      7081303.13      2837002.79      7080545.77
      2838174.63      7080098.43      2838642.76      7079526.36
      2839255.80      7079411.15      2839743.42      7078503.88
      2840311.55      7078128.22      2840728.33      7077102.58
      2842150.88      7076013.44      2842379.15      7075152.26
      2842944.79      7074347.37      2843348.27      7073903.38
      2843947.22      7073729.27      2844385.55      7073180.67

Type RM Length L Ch R = 1,27004,402,402,402
BEGIN DESCRIPTION:
CHAFFIN CREEK 44.0
END DESCRIPTION:
XS GIS Cut Line= 3
      2831575.01      7089225.01      2831275.00      7089025.00
      2830975.01      7088975.00
#Sta/Elev= 30
  4643.5  531.70  4759.2  521.60  4795.2  518.97  4867.4  515.74  4915.0  514.53
  4958.1  514.26  4975.5  513.84  4981.5  512.90  4990.5  509.32  4996.6  508.31
  4998.1  504.61  4998.6  503.81  5003.6  503.81  5004.1  504.61  5006.6  504.61
  5014.2  510.70  5024.3  511.80  5031.9  512.18  5064.9  511.11  5075.0  511.68
  5092.8  510.68  5097.8  508.24  5105.4  511.09  5115.6  511.57  5135.9  514.01
  5147.5  514.53  5186.6  515.59  5206.8  516.77  5247.4  521.15  5308.2  525.85
#Mann=4,-1,0
  4643.5    0.05       0  4958.1    0.12       0  4998.1    0.07       0
  5004.1    0.12       0
Bank Sta=4915,5147.5
Exp/Cntr=0.3,0.1

Type RM Length L Ch R = 1,26602,612,612,612
BEGIN DESCRIPTION:
CHAFFIN CREEK 43.0
END DESCRIPTION:
XS GIS Cut Line= 3
      2831604.81      7089176.91      2831222.60      7088799.16
      2830975.04      7088725.01
#Sta/Elev= 30
  4464.4  531.36  4628.3  519.11  4699.0  516.06  4763.7  515.18  4779.8  513.84
  4798.0  510.35  4812.1  509.67  4819.2  511.38  4833.3  510.07  4840.4  512.89
  4847.4  513.25  4861.6  512.42  4932.3  512.18  4967.7  513.11  4981.8  511.18
  4988.9  504.80  4993.0  504.07  4993.5  503.27  4998.5  503.27  4999.0  504.07
  5001.2  506.61  5009.7  509.29  5029.5  512.20  5032.1  513.84  5034.8  515.59
  5041.0  516.37  5061.9  517.29  5067.8  518.72  5128.9  523.92  5260.2  530.75
#Mann=5,-1,0
  4464.4    0.05       0  4763.7    0.12       0  4993.0    0.07       0
  4999.0    0.12       0  5128.9    0.05       0
Bank Sta=4779.8,5032.1
Exp/Cntr=0.3,0.1

Type RM Length L Ch R = 1,25990,337,337,337
BEGIN DESCRIPTION:
CHAFFIN CREEK 42.0
END DESCRIPTION:
XS GIS Cut Line= 3
      2831824.96      7088824.98      2831564.60      7088711.99
      2831075.02      7088575.01
#Sta/Elev= 30
  4723.6  530.62  4799.9  529.23  4837.3  527.47  4919.8  522.00  4960.0  520.71
  4965.5  520.28  4974.3  517.88  4984.4  511.73  4989.0  508.94  4991.4  505.36
  4993.1  502.83  4993.6  502.03  4998.6  502.03  4999.1  502.83  5009.8  503.38
  5013.5  507.90  5047.6  511.35  5110.8  510.53  5178.4  511.08  5233.4  511.73
  5328.9  513.77  5346.6  515.19  5351.8  514.92  5386.0  516.65  5420.1  519.67
  5425.3  519.50  5459.4  523.19  5493.6  524.52  5498.8  524.16  5515.8  525.37
#Mann=5,-1,0
  4723.6    0.05       0  4991.4    0.16       0  4993.1    0.07       0
  4999.1    0.16       0  5178.4    0.05       0
Bank Sta=4984.4,5233.4
Exp/Cntr=0.3,0.1

Type RM Length L Ch R = 1,25653,250,250,250
BEGIN DESCRIPTION:
CHAFFIN CREEK 41.0
END DESCRIPTION:
XS GIS Cut Line= 3
      2831843.42      7088604.77      2831525.00      7088525.00
      2831074.96      7088525.00
#Sta/Elev= 30
  4649.5  525.31  4715.4  522.55  4872.2  514.58  4905.6  512.07  4913.4  510.30
  4916.5  510.79  4946.8  510.45  4952.5  509.78  4959.7  510.37  4980.3  508.74
  4987.8  506.72  4994.8  501.18  4995.3  500.38  5000.3  500.38  5000.8  501.18
  5002.8  502.48  5017.8  507.49  5027.8  507.02  5037.8  508.21  5057.8  508.35
  5078.5  509.78  5099.5  510.88  5177.8  511.46  5207.8  512.49  5367.8  521.26
  5397.8  521.97  5407.8  523.49  5417.8  527.70  5425.3  529.74  5427.8  529.74
#Mann=6,-1,0
  4649.5    0.05       0  4715.4    0.16       0  4916.5    0.12       0
  4994.8    0.07       0  5000.8    0.12       0  5099.5    0.05       0
Bank Sta=4952.5,5078.5
Exp/Cntr=0.3,0.1

Type RM Length L Ch R = 1,25403,430,430,430
BEGIN DESCRIPTION:
Mapping XS d32e3329
END DESCRIPTION:
XS GIS Cut Line= 3
      2831897.69      7088522.00      2831533.31      7088327.51
      2831272.83      7088209.52
#Sta/Elev= 30
  4581.4  523.72  4637.2  521.06  4692.0  517.44  4765.8  515.25  4818.0  512.72
  4840.0  510.63  4856.3  510.10  4862.2  508.84  4867.8  505.93  4878.2  505.40
  4913.2  506.57  4935.8  505.42  4958.5  505.44  4966.1  505.65  4981.2  509.80
  4988.0  506.58  4988.8  500.56  4989.3  499.76  4994.3  499.76  4994.8  500.56
  5003.6  502.09  5010.8  505.30  5016.3  506.78  5025.5  507.58  5039.4  506.88
  5069.5  508.74  5071.8  508.85  5108.7  511.30  5223.1  514.90  5280.4  519.67
#Mann=5,-1,0
  4581.4    0.05       0  4637.2    0.16       0  4988.8    0.07       0
  4994.8    0.16       0  5069.5    0.05       0
Bank Sta=4862.2,5071.8
Exp/Cntr=0.3,0.1

Type RM Length L Ch R = 1,24973,288,288,288
BEGIN DESCRIPTION:
CHAFFIN CREEK 40.0
END DESCRIPTION:
XS GIS Cut Line= 3
      2832075.01      7088425.01      2831725.00      7088125.00
      2831274.97      7088024.99
#Sta/Elev= 30
  4536.4  528.84  4592.9  526.32  4757.4  514.26  4891.5  507.71  4912.3  506.03
  4969.4  506.55  4978.8  505.23  4983.7  504.30  4990.3  500.86  4991.1  497.93
  4991.6  497.13  4996.6  497.13  4997.1  497.93  5000.0  497.93  5007.6  502.10
  5016.6  502.55  5021.7  506.00  5038.4  504.05  5051.8  505.23  5070.4  507.78
  5079.3  507.74  5099.8  510.02  5119.7  510.43  5222.8  512.04  5293.2  514.15
  5341.8  519.23  5390.5  522.93  5407.2  525.44  5434.0  527.67  5458.4  528.57
#Mann=5,-1,0
  4536.4    0.05       0  4757.4    0.16       0  4991.1    0.07       0
  4997.1    0.16       0  5119.7    0.05       0
Bank Sta=4978.8,5051.8
Exp/Cntr=0.3,0.1

Type RM Length L Ch R = 1,24685,466,466,466
BEGIN DESCRIPTION:
CHAFFIN CREEK 39.0
END DESCRIPTION:
XS GIS Cut Line= 3
      2832203.89      7088090.57      2831920.02      7087949.75
      2831412.59      7087777.63
#Sta/Elev= 30
  4667.0  517.36  4669.8  516.67  4731.5  515.50  4877.9  506.03  4910.8  505.93
  4912.9  505.19  4916.4  503.93  4922.5  505.55  4933.2  505.07  4938.8  504.12
  4961.2  503.92  4967.2  502.04  4978.0  501.79  4983.6  498.81  4986.2  496.34
  4986.7  495.54  4991.7  495.54  4992.2  496.34  4999.7  497.39  5009.6  501.14
  5014.0  505.19  5014.9  506.06  5046.3  507.68  5135.2  506.87  5179.3  508.16
  5229.5  510.83  5379.9  515.95  5386.5  517.08  5401.0  517.88  5519.7  522.22
#Mann=3,-1,0
  4667.0    0.05       0  4986.2    0.03       0  4992.2    0.05       0
Bank Sta=4912.9,5014
Exp/Cntr=0.3,0.1

Type RM Length L Ch R = 1,24219,457,457,457
BEGIN DESCRIPTION:
Mapping XS 3ad40651
END DESCRIPTION:
XS GIS Cut Line= 3
      2832441.05      7087900.97      2831782.20      7087588.48
      2831514.02      7087591.08
#Sta/Elev= 30
  4253.7  515.62  4351.9  510.73  4442.8  508.83  4481.8  506.86  4511.0  507.77
  4516.6  506.99  4533.8  507.59  4624.7  506.42  4653.0  507.11  4658.8  506.72
  4667.9  504.52  4675.5  503.98  4698.5  503.80  4721.2  506.45  4831.4  505.92
  4885.9  506.35  4968.7  505.25  4981.1  501.97  4990.1  496.68  4997.1  494.55
  4997.6  493.75  5002.7  493.75  5003.2  494.55  5010.1  497.95  5017.0  504.52
  5030.1  515.79  5039.7  520.23  5070.4  522.92  5142.5  525.79  5251.1  526.97
#Mann=7,-1,0
  4253.7    0.05       0  4675.5    0.16       0  4831.4    0.12       0
  4997.1    0.07       0  5003.2    0.12       0  5039.7    0.16       0
  5070.4    0.05       0
Bank Sta=4667.9,5017
Exp/Cntr=0.3,0.1

Type RM Length L Ch R = 1,23762,599,599,599
BEGIN DESCRIPTION:
double CHAFFIN CREEK 38.0
END DESCRIPTION:
XS GIS Cut Line= 3
      2832625.05      7087275.00      2832075.00      7087325.00
      2831624.98      7087275.00
#Sta/Elev= 30
  4450.8  538.55  4511.1  532.26  4561.3  524.48  4665.0  513.16  4701.9  506.93
  4732.5  504.68  4755.1  503.30  4772.2  497.65  4782.2  502.02  4802.3  503.67
  4882.6  503.22  4922.8  504.38  4942.9  501.56  4952.9  502.04  4973.0  501.44
  4983.0  499.13  4990.0  493.32  4990.5  492.52  4996.1  493.32  5005.6  493.88
  5013.2  498.39  5023.2  501.96  5073.5  501.71  5079.6  503.30  5093.7  505.09
  5133.9  505.34  5184.2  508.53  5251.3  514.25  5355.3  523.06  5455.9  527.40
#Mann=7,-1,0
  4450.8    0.16       0  4665.0    0.12       0  4732.5    0.16       0
  4952.9    0.12       0  4990.0    0.07       0  4996.1    0.12       0
  5251.3    0.16       0
Bank Sta=4755.1,5079.6
Exp/Cntr=0.3,0.1

Type RM Length L Ch R = 1,23163,243,243,243
BEGIN DESCRIPTION:
CHAFFIN CREEK 37.0
END DESCRIPTION:
XS GIS Cut Line= 3
      2832675.00      7087125.00      2832275.00      7086875.00
      2831674.96      7087025.01
#Sta/Elev= 30
  4528.3  539.31  4578.4  531.20  4609.1  527.86  4615.0  528.23  4694.0  518.29
  4730.5  515.17  4752.4  514.69  4767.1  511.98  4816.8  507.73  4888.5  504.50
  4931.9  502.70  4942.5  501.46  4964.6  502.92  4977.0  501.57  4986.4  494.22
  4992.3  494.20  4993.9  490.39  4994.4  489.59  5000.2  490.39  5002.6  490.39
  5010.3  495.93  5018.0  499.54  5023.2  498.35  5030.9  500.30  5059.3  499.33
  5081.8  501.46  5247.4  502.49  5329.8  504.88  5383.7  508.21  5618.5  526.55
#Mann=7,-1,0
  4528.3    0.16       0  4816.8    0.05       0  4888.5    0.16       0
  4931.9    0.12       0  4993.9    0.07       0  5000.2    0.12       0
  5383.7    0.16       0
Bank Sta=4942.5,5081.8
Exp/Cntr=0.3,0.1

Type RM Length L Ch R = 1,22920,365,365,365
BEGIN DESCRIPTION:
Mapping XS ccdb3b85
END DESCRIPTION:
XS GIS Cut Line= 3
      2832608.59      7086758.62      2832226.65      7086650.98
      2831838.93      7086630.21
#Sta/Elev= 30
  4592.2  531.15  4606.3  529.16  4622.9  524.55  4628.1  524.92  4647.9  520.42
  4689.4  513.36  4696.2  510.76  4720.6  507.86  4762.2  505.37  4873.2  503.09
  4918.7  502.10  4950.0  500.71  4980.3  497.40  4987.3  494.31  4992.4  494.31
  4997.5  489.40  4998.0  488.60  5003.3  488.60  5003.8  489.40  5011.5  492.97
  5020.7  499.39  5030.7  500.48  5090.8  501.27  5110.8  498.92  5150.9  499.21
  5166.6  500.71  5188.8  503.75  5251.0  510.17  5291.1  513.13  5377.3  516.22
#Mann=6,-1,0
  4592.2    0.05       0  4873.2    0.16       0  4918.7    0.12       0
  4997.5    0.07       0  5003.8    0.12       0  5188.8    0.16       0
Bank Sta=4950,5166.6
Exp/Cntr=0.3,0.1

Type RM Length L Ch R = 1,22555,701,701,701
BEGIN DESCRIPTION:
CHAFFIN CREEK 36.0
END DESCRIPTION:
XS GIS Cut Line= 3
      2832716.27      7086473.91      2832375.00      7086375.00
      2831925.00      7086125.00
#Sta/Elev= 30
  4654.6  531.38  4664.9  531.06  4697.6  524.90  4760.0  510.93  4776.0  508.53
  4781.2  509.22  4835.7  503.77  4852.4  499.57  4905.8  497.68  4938.2  498.17
  4978.7  499.24  4987.9  493.56  4993.1  491.91  4996.3  487.73  4996.8  486.93
  5002.3  486.93  5002.8  487.73  5007.3  491.01  5012.8  491.01  5017.9  494.77
  5032.8  498.00  5043.5  498.37  5055.7  499.96  5131.7  499.57  5215.8  499.80
  5310.8  501.22  5364.5  505.25  5376.0  507.23  5435.5  513.13  5524.7  520.21
#Mann=6,-1,0
  4654.6    0.05       0  4835.7    0.16       0  4938.2    0.12       0
  4996.3    0.07       0  5002.8    0.12       0  5043.5    0.16       0
Bank Sta=4852.4,5131.7
Exp/Cntr=0.3,0.1

Type RM Length L Ch R = 1,21854,240,240,240
BEGIN DESCRIPTION:
CHAFFIN CREEK 35.0
END DESCRIPTION:
XS GIS Cut Line= 3
      2832924.99      7086125.00      2832475.00      7085975.00
      2831925.05      7086074.99
#Sta/Elev= 30
  4544.0  537.59  4607.2  534.89  4681.0  528.63  4744.3  522.19  4860.2  508.38
  4891.8  506.54  4937.0  500.77  4944.5  499.68  4965.6  499.47  4974.2  497.12
  4976.2  496.57  4986.7  486.80  4994.0  485.67  4994.5  484.87  5000.0  484.87
  5000.5  485.67  5007.8  492.11  5015.7  495.10  5050.1  495.17  5070.0  497.12
  5079.3  499.22  5176.4  498.29  5273.7  497.44  5333.4  498.82  5385.5  502.28
  5433.8  507.73  5438.9  507.51  5445.2  508.97  5492.2  514.02  5577.3  520.16
#Mann=5,-1,0
  4544.0    0.05       0  4937.0    0.12       0  4994.0    0.07       0
  5000.5    0.12       0  5176.4    0.16       0
Bank Sta=4974.2,5070
Exp/Cntr=0.3,0.1

Type RM Length L Ch R = 1,21614,814,814,814
BEGIN DESCRIPTION:
Mapping XS 18d68781
END DESCRIPTION:
XS GIS Cut Line= 3
      2832948.01      7085759.48      2832531.33      7085768.16
      2831980.83      7085950.22
#Sta/Elev= 30
  4575.2  534.27  4698.2  526.60  4928.3  504.64  4965.6  499.54  4984.1  496.34
  4992.0  495.51  4995.6  490.16  5000.9  485.85  5005.9  485.15  5006.4  484.35
  5012.4  485.15  5032.6  495.29  5104.0  493.73  5122.5  498.06  5191.2  497.12
  5198.8  496.57  5209.3  493.73  5221.6  494.86  5230.4  497.55  5293.6  497.37
  5312.8  493.93  5323.0  496.34  5356.8  496.98  5430.5  501.12  5445.0  502.89
  5471.4  508.94  5476.7  508.55  5483.1  510.46  5503.2  512.72  5571.8  514.34
#Mann=5,-1,0
  4575.2    0.05       0  4965.6    0.12       0  5005.9    0.07       0
  5012.4    0.12       0  5221.6    0.16       0
Bank Sta=4984.1,5323
Exp/Cntr=0.3,0.1

Type RM Length L Ch R = 1,20800,526,526,526
BEGIN DESCRIPTION:
CHAFFIN CREEK 34.0
END DESCRIPTION:
XS GIS Cut Line= 3
      2832875.02      7085575.01      2832425.00      7085425.00
      2831868.62      7085338.69
#Sta/Elev= 30
  4526.9  526.65  4543.3  525.92  4579.6  525.22  4664.0  520.98  4695.6  518.16
  4748.3  511.33  4811.5  504.97  4853.7  501.73  4948.6  496.92  4969.0  493.39
  4980.2  490.07  4987.4  481.66  4987.9  480.86  4993.5  480.86  4994.0  481.66
  4998.6  482.96  5003.8  482.96  5021.5  491.70  5030.2  492.51  5103.3  491.97
  5126.6  493.39  5142.9  495.41  5153.1  495.87  5297.3  495.97  5375.7  497.85
  5406.0  500.16  5456.6  505.34  5491.3  507.73  5559.3  514.06  5564.3  515.07
#Mann=4,-1,0
  4526.9    0.08       0  4543.3    0.16       0  4987.4    0.07       0
  4994.0    0.12       0
Bank Sta=4969,5126.6
Exp/Cntr=0.3,0.1

Type RM Length L Ch R = 1,20274,135,135,135
BEGIN DESCRIPTION:
Mapping XS 93c0d4b8
END DESCRIPTION:
XS GIS Cut Line= 5
      2832839.49      7085342.79      2832817.79      7085099.76
      2832518.31      7084982.57      2832127.69      7084956.53
      2831832.59      7085056.35
#Sta/Elev= 30
  4419.0  520.28  4529.0  516.82  4597.5  516.11  4708.9  511.72  4775.4  507.38
  4829.7  501.11  4884.0  496.65  4908.5  496.15  4929.4  494.24  4958.4  491.90
  4977.4  485.80  4983.7  482.87  4988.8  482.87  4994.6  480.07  4995.1  479.27
  5000.7  479.27  5001.2  480.07  5008.0  482.64  5018.0  490.95  5020.3  491.90
  5028.1  493.16  5078.1  492.49  5308.6  494.68  5400.0  496.81  5417.0  498.55
  5505.6  501.57  5542.7  505.69  5631.8  511.01  5642.8  512.75  5687.6  514.63
#Mann=4,-1,0
  4419.0    0.16       0  4929.4    0.12       0  4994.6    0.07       0
  5001.2    0.12       0
Bank Sta=4958.4,5020.3
Exp/Cntr=0.3,0.1

Type RM Length L Ch R = 1,20139,389,389,389
BEGIN DESCRIPTION:
Mapping XS b431fa07
END DESCRIPTION:
XS GIS Cut Line= 4
      2832982.71      7085052.01      2832817.79      7084904.45
      2832422.83      7084835.00      2831889.51      7084761.29
#Sta/Elev= 30
  4506.9  516.91  4602.2  514.56  4638.0  508.80  4673.2  506.19  4687.4  506.34
  4694.1  508.29  4701.6  507.19  4708.3  509.51  4715.8  507.92  4722.5  508.85
  4809.4  501.31  4870.6  497.57  4934.1  495.13  4962.0  491.46  4970.8  489.00
  4982.3  485.39  4991.7  479.92  4992.2  479.12  4997.8  479.12  4998.3  479.92
  5005.2  481.93  5015.3  489.02  5025.5  491.58  5046.7  490.64  5061.9  491.29
  5064.2  491.46  5270.6  492.99  5440.0  495.97  5561.1  507.20  5667.6  512.69
#Mann=7,-1,0
  4506.9    0.05       0  4870.6    0.16       0  4970.8    0.12       0
  4991.7    0.07       0  4998.3    0.12       0  5061.9    0.16       0
  5270.6    0.05       0
Bank Sta=4962,5064.2
Exp/Cntr=0.3,0.1

Type RM Length L Ch R = 1,19750,247,247,247
BEGIN DESCRIPTION:
Mapping XS 0ed86a9f
END DESCRIPTION:
XS GIS Cut Line= 3
      2833039.15      7084864.52      2832820.40      7084619.73
      2832112.04      7084390.55
#Sta/Elev= 30
  4651.6  516.43  4753.5  515.17  4796.1  513.32  4810.3  512.20  4873.8  505.63
  4909.0  501.09  4923.2  499.67  4961.6  496.94  4965.8  496.58  4972.8  492.18
  4979.7  490.47  4980.1  489.90  4985.6  481.06  4992.8  479.20  4993.3  478.40
  4998.9  478.40  4999.4  479.20  5011.7  481.21  5017.1  484.88  5027.6  488.65
  5043.7  489.89  5069.6  489.45  5080.3  489.90  5122.2  490.69  5209.0  490.61
  5353.4  491.85  5574.1  494.99  5630.3  496.76  5710.8  500.60  5724.4  500.69
#Mann=5,-1,0
  4651.6    0.05       0  4961.6    0.12       0  4992.8    0.07       0
  4999.4    0.12       0  5353.4    0.16       0
Bank Sta=4980.1,5080.3
Exp/Cntr=0.3,0.1

Type RM Length L Ch R = 1,19503,819,819,819
BEGIN DESCRIPTION:
Mapping XS 01428445
END DESCRIPTION:
XS GIS Cut Line= 3
      2833080.80      7084812.41      2832888.10      7084406.19
      2832195.40      7084041.60
#Sta/Elev= 30
  4537.1  514.00  4681.3  513.49  4817.7  496.87  4871.7  493.11  4914.2  491.38
  4929.4  489.18  4965.9  488.70  4982.4  483.90  4984.6  479.18  4994.6  478.84
  4995.1  478.04  5001.3  478.84  5016.1  487.26  5020.0  488.76  5025.6  483.66
  5035.4  487.98  5042.0  487.64  5047.7  484.68  5064.0  485.41  5069.7  481.61
  5080.4  483.02  5086.1  487.75  5107.7  489.02  5113.7  489.18  5271.2  490.26
  5388.9  491.21  5537.5  494.95  5581.6  497.64  5669.7  506.01  5769.5  512.09
#Mann=7,-1,0
  4537.1    0.05       0  4871.7    0.12       0  4994.6    0.07       0
  5001.3    0.12       0  5016.1    0.16       0  5107.7    0.12       0
  5271.2    0.16       0
Bank Sta=4929.4,5113.7
Exp/Cntr=0.3,0.1

Type RM Length L Ch R = 1,18684,559,559,559
BEGIN DESCRIPTION:
CHAFFIN CREEK 30.0
END DESCRIPTION:
XS GIS Cut Line= 3
      2833575.01      7084425.02      2833325.00      7083975.00
      2832575.04      7083525.02
#Sta/Elev= 30
  4497.7  511.58  4600.7  502.38  4668.2  495.18  4673.9  495.62  4711.6  492.41
  4822.3  486.50  4844.5  485.48  4895.8  484.88  4939.3  485.59  4945.0  485.14
  4955.3  482.33  4966.7  483.16  4982.8  481.63  4989.6  478.07  4995.3  476.96
  4995.8  476.16  5001.7  476.16  5002.2  476.96  5009.6  485.32  5020.3  486.24
  5222.4  484.90  5307.9  486.50  5445.0  488.27  5523.7  490.68  5587.8  495.84
  5661.3  500.19  5747.2  507.07  5762.8  509.13  5778.3  509.32  5887.1  517.19
#Mann=6,-1,0
  4497.7    0.16       0  4844.5    0.12       0  4995.3    0.07       0
  5002.2    0.12       0  5445.0    0.16       0  5661.3    0.05       0
Bank Sta=4822.3,5307.9
Exp/Cntr=0.3,0.1

Type RM Length L Ch R = 1,18125,535,535,535
BEGIN DESCRIPTION:
CHAFFIN CREEK 29.0
END DESCRIPTION:
XS GIS Cut Line= 3
      2833875.00      7084425.01      2833675.00      7083675.00
      2833124.97      7083424.99
#Sta/Elev= 30
  4277.4  514.94  4369.9  504.61  4472.4  497.12  4577.5  488.01  4715.3  484.14
  4765.4  483.42  4888.0  483.00  4929.4  484.43  4977.1  483.04  4977.4  482.98
  4981.2  482.29  4992.6  474.08  4993.1  473.28  4999.5  474.08  5012.2  481.43
  5036.1  483.45  5051.0  481.82  5075.6  483.41  5145.1  482.31  5160.2  481.87
  5165.7  479.77  5206.3  482.05  5218.4  479.77  5263.4  483.85  5289.9  482.98
  5353.3  483.97  5493.0  488.89  5522.7  491.81  5580.9  500.65  5657.8  506.77
#Mann=9,-1,0
  4277.4    0.16       0  4472.4    0.05       0  4715.3    0.07       0
  4765.4    0.05       0  4977.1    0.12       0  4992.6    0.07       0
  4999.5    0.12       0  5145.1    0.16       0  5353.3    0.05       0
Bank Sta=4977.4,5289.9
Exp/Cntr=0.3,0.1

Type RM Length L Ch R = 1,17590,717,717,717
BEGIN DESCRIPTION:
CHAFFIN CREEK 28.0
END DESCRIPTION:
XS GIS Cut Line= 3
      2833925.00      7084324.96      2834025.00      7083525.00
      2833924.99      7083074.97
#Sta/Elev= 30
  4170.9  506.29  4238.9  499.48  4312.0  494.33  4342.2  490.64  4432.9  485.14
  4581.0  481.97  4755.9  482.36  4854.2  481.43  4896.5  480.67  4934.3  482.44
  4939.3  481.90  4967.0  472.01  4970.9  471.99  4971.5  471.19  4978.2  471.99
  5018.1  473.03  5034.5  481.97  5038.6  484.06  5045.0  484.86  5088.5  487.21
  5151.2  496.31  5184.0  499.77  5202.5  501.00  5227.5  500.58  5331.7  494.45
  5345.9  494.81  5365.1  492.54  5370.2  493.52  5386.8  491.09  5438.1  492.98
#Mann=9,-1,0
  4170.9    0.16       0  4238.9    0.05       0  4755.9    0.16       0
  4854.2    0.12       0  4970.9    0.07       0  4978.2    0.12       0
  5184.0    0.16       0  5227.5    0.12       0  5331.7    0.16       0
Bank Sta=4581,5034.5
Exp/Cntr=0.3,0.1

Type RM Length L Ch R = 1,16873,419,419,419
BEGIN DESCRIPTION:
CHAFFIN CREEK 27.0
END DESCRIPTION:
XS GIS Cut Line= 3
      2834987.07      7083979.11      2834565.19      7083307.23
      2834253.55      7083099.47
#Sta/Elev= 30
  4176.4  504.69  4203.7  502.51  4209.6  503.13  4224.9  500.53  4246.2  499.56
  4252.1  498.29  4298.0  494.29  4413.4  486.88  4544.2  481.78  4663.6  479.66
  4681.3  479.51  4753.9  477.70  4948.8  479.23  4972.9  476.70  4979.4  475.09
  4985.4  475.70  4996.5  470.41  4997.1  469.61  5003.7  469.61  5004.4  470.41
  5015.4  474.98  5021.5  479.05  5092.0  478.67  5107.9  479.66  5144.6  482.40
  5174.3  485.93  5201.7  490.73  5216.8  491.44  5282.5  498.29  5344.3  500.11
#Mann=5,-1,0
  4176.4    0.05       0  4681.3    0.12       0  4996.5    0.07       0
  5004.4    0.12       0  5092.0    0.16       0
Bank Sta=4663.6,5107.9
Exp/Cntr=0.3,0.1

Type RM Length L Ch R = 1,16454,535,535,535
BEGIN DESCRIPTION:
CHAFFIN CREEK 26.0
END DESCRIPTION:
XS GIS Cut Line= 3
      2835374.97      7083324.98      2834725.00      7082925.00
      2834424.97      7082574.97
#Sta/Elev= 30
  4222.8  509.56  4352.3  500.32  4441.1  497.66  4499.1  493.76  4535.8  491.11
  4563.3  487.69  4599.6  485.42  4651.7  480.09  4760.7  475.66  4761.4  475.64
  4788.9  475.26  4833.3  477.11  4864.9  477.24  4978.3  477.81  4983.0  470.59
  5003.4  469.81  5004.1  469.01  5010.7  469.01  5011.3  469.81  5014.0  474.93
  5021.7  474.17  5024.8  475.64  5028.2  477.29  5035.9  477.90  5099.6  476.16
  5206.0  480.85  5255.4  486.10  5269.7  486.57  5333.4  497.10  5447.0  503.36
#Mann=5,-1,0
  4222.8    0.05       0  4760.7    0.16       0  4864.9    0.05       0
  5003.4    0.03       0  5011.3    0.05       0
Bank Sta=4761.4,5024.8
Exp/Cntr=0.3,0.1

Type RM Length L Ch R = 1,15919,404,404,404
BEGIN DESCRIPTION:
CHAFFIN CREEK 25.0
END DESCRIPTION:
XS GIS Cut Line= 3
      2835725.01      7083175.01      2834925.00      7082425.00
      2834425.00      7082425.00
#Sta/Elev= 30
  3871.5  514.96  3885.4  514.90  3892.8  513.56  3899.6  513.91  4161.4  497.23
  4203.9  492.89  4288.9  487.25  4296.2  485.70  4338.2  482.26  4525.7  475.09
  4642.6  473.94  4664.0  471.93  4670.9  472.07  4678.2  473.98  4699.2  474.37
  4819.4  473.87  4961.0  476.04  4970.6  475.75  4978.1  472.99  4984.1  466.94
  4984.8  466.14  4992.0  466.94  4998.1  467.21  5008.1  470.07  5018.1  475.27
  5038.1  475.82  5108.1  473.33  5142.2  475.09  5278.1  490.84  5468.1  506.32
#Mann=3,-1,0
  3871.5    0.05       0  4984.1    0.03       0  4992.0    0.05       0
Bank Sta=4525.7,5142.2
Exp/Cntr=0.3,0.1

Type RM Length L Ch R = 1,15515,179,179,179
BEGIN DESCRIPTION:
Mapping XS b0f8d691
END DESCRIPTION:
XS GIS Cut Line= 3
      2835658.93      7083031.17      2835153.73      7082140.56
      2834877.88      7081609.67
#Sta/Elev= 30
  3969.2  506.62  4033.8  501.42  4080.6  499.33  4173.6  491.19  4394.3  482.98
  4459.2  477.86  4565.9  474.42  4658.2  472.18  4674.1  473.45  4679.9  472.08
  4695.8  473.62  4739.0  471.24  4754.9  473.01  4975.6  474.11  4981.3  473.70
  4987.7  466.92  4993.5  466.10  4994.1  465.30  5001.5  466.10  5010.7  472.62
  5019.6  474.42  5091.6  473.76  5108.0  471.08  5135.8  471.65  5166.5  474.42
  5345.7  480.24  5412.0  484.84  5434.1  483.80  5494.8  484.77  5591.4  494.54
#Mann=4,-1,0
  3969.2    0.05       0  4080.6    0.08       0  4993.5    0.07       0
  5001.5    0.08       0
Bank Sta=4565.9,5166.5
Exp/Cntr=0.3,0.1

Type RM Length L Ch R = 1,15336,457,457,457
BEGIN DESCRIPTION:
Mapping XS 78fb4895
END DESCRIPTION:
XS GIS Cut Line= 3
      2835799.54      7082968.64      2835268.31      7082005.14
      2834977.09      7081459.09
#Sta/Elev= 30
  3894.4  505.25  3966.3  501.20  4077.7  495.61  4208.4  487.48  4242.4  486.37
  4305.8  483.86  4349.4  483.76  4392.9  479.10  4532.1  474.78  4630.0  473.35
  4755.0  471.86  4968.3  473.43  4974.1  472.96  4983.4  470.34  4988.8  465.34
  4989.5  464.54  4996.2  464.54  4996.9  465.34  5006.1  466.38  5017.7  473.49
  5030.7  473.51  5104.1  473.35  5177.2  475.93  5291.4  482.97  5316.2  485.07
  5330.1  486.89  5412.3  490.00  5516.1  490.67  5595.1  496.96  5613.5  498.39
#Mann=11,-1,0
  3894.4    0.08       0  3966.3    0.05       0  4242.4    0.08       0
  4532.1    0.05       0  4988.8    0.03       0  4996.9    0.05       0
  5030.7    0.08       0  5177.2    0.05       0  5291.4     0.1       0
  5316.2    0.08       0  5595.1    0.05       0
Bank Sta=4630,5104.1
Exp/Cntr=0.3,0.1

Type RM Length L Ch R = 1,14879,517,517,517
BEGIN DESCRIPTION:
CHAFFIN CREEK 23.0
END DESCRIPTION:
XS GIS Cut Line= 3
      2836024.99      7082474.97      2835625.00      7081725.00
      2835374.98      7081324.97
#Sta/Elev= 30
  4131.9  502.44  4154.5  498.94  4310.0  486.70  4337.6  482.75  4378.1  481.33
  4414.1  479.07  4436.1  479.94  4528.6  475.27  4562.2  475.38  4665.0  471.51
  4709.9  470.29  4759.8  471.93  4885.9  471.15  4959.2  472.44  4968.1  471.44
  4979.0  464.56  4985.5  464.50  4986.2  463.70  4993.6  464.50  5010.8  471.13
  5017.2  471.81  5040.8  471.09  5047.3  468.78  5053.2  471.32  5086.1  471.51
  5105.1  474.49  5162.9  478.99  5287.9  483.98  5372.8  490.85  5453.6  495.03
#Mann=5,-1,0
  4131.9    0.05       0  4378.1    0.08       0  4528.6    0.05       0
  4985.5    0.03       0  4993.6    0.05       0
Bank Sta=4665,5086.1
Exp/Cntr=0.3,0.1

Type RM Length L Ch R = 1,14362,179,179,179
BEGIN DESCRIPTION:
Mapping XS e99154f3
END DESCRIPTION:
XS GIS Cut Line= 3
      2835952.34      7082140.58      2835959.29      7081376.67
      2835990.48      7080919.17
#Sta/Elev= 30
  4226.0  481.89  4239.0  479.65  4271.6  480.19  4321.6  479.14  4341.6  477.15
  4630.2  472.10  4634.8  471.99  4891.6  468.93  4961.6  470.87  4971.6  470.46
  4984.2  462.48  4984.9  461.68  4992.4  462.48  4998.5  464.80  5003.6  462.99
  5021.7  469.81  5031.7  470.28  5081.8  463.87  5091.8  464.74  5111.9  470.87
  5121.9  470.28  5131.9  465.80  5147.2  469.99  5152.2  468.16  5162.0  469.65
  5217.2  470.63  5245.4  471.99  5372.5  482.42  5412.6  488.78  5448.5  490.31
#Mann=6,-1,0
  4226.0    0.05       0  4239.0    0.08       0  4630.2    0.05       0
  4984.2    0.04       0  4992.4    0.05       0  5217.2    0.08       0
Bank Sta=4634.8,5245.4
Exp/Cntr=0.3,0.1

Type RM Length L Ch R = 1,14183,462,462,462
BEGIN DESCRIPTION:
Mapping XS ead6376c
END DESCRIPTION:
XS GIS Cut Line= 3
      2836056.51      7082161.36      2836059.98      7081275.98
      2836080.81      7080880.11
#Sta/Elev= 30
  4088.6  486.78  4119.9  485.51  4175.0  484.27  4195.0  479.85  4315.5  479.79
  4445.0  474.53  4587.3  471.87  4825.0  469.56  4974.0  470.76  4977.2  470.59
  4990.6  461.67  4991.4  460.87  4998.5  460.87  4999.3  461.67  5005.0  462.56
  5015.0  467.59  5025.0  470.29  5055.1  469.35  5065.1  470.08  5075.1  467.84
  5085.1  464.14  5105.1  464.19  5115.2  464.57  5135.2  469.08  5145.2  464.86
  5162.4  470.49  5193.7  471.87  5295.4  480.37  5335.5  480.41  5370.4  478.38
#Mann=5,-1,0
  4088.6    0.05       0  4119.9    0.08       0  4315.5    0.12       0
  4990.6    0.07       0  4999.3    0.12       0
Bank Sta=4587.3,5193.7
Exp/Cntr=0.3,0.1

Type RM Length L Ch R = 1,13721,736,736,736
BEGIN DESCRIPTION:
Mapping XS 3f89ab82
END DESCRIPTION:
XS GIS Cut Line= 3
      2836445.40      7081741.29      2836362.06      7081175.28
      2836330.82      7080640.60
#Sta/Elev= 30
  4407.9  485.88  4442.3  485.22  4447.3  484.27  4464.8  484.61  4495.1  483.27
  4512.0  483.38  4517.0  482.25  4525.4  481.88  4642.7  478.97  4808.2  471.02
  4879.2  467.99  4919.6  469.56  4960.1  468.49  4970.2  467.73  4977.6  465.51
  4982.7  465.51  4995.9  460.08  4996.7  459.28  5004.0  459.28  5004.8  460.08
  5010.3  462.07  5015.4  466.36  5020.4  468.85  5030.4  469.34  5110.5  467.51
  5310.9  470.61  5357.1  470.13  5412.3  471.02  5441.1  473.47  5515.6  475.40
#Mann=4,-1,0
  4407.9    0.05       0  4642.7    0.12       0  4995.9    0.07       0
  5004.8    0.12       0
Bank Sta=4808.2,5412.3
Exp/Cntr=0.3,0.1

Type RM Length L Ch R = 1,12985,528,528,528
BEGIN DESCRIPTION:
CHAFFIN CREEK 20.0
END DESCRIPTION:
XS GIS Cut Line= 3
      2836903.55      7081383.69      2836660.49      7080965.42
      2836391.52      7080570.60
#Sta/Elev= 30
  4515.2  489.83  4524.6  489.02  4594.7  484.38  4616.9  481.12  4638.4  480.06
  4644.2  481.75  4675.6  479.48  4697.2  476.67  4703.0  473.90  4718.7  472.90
  4746.0  474.22  4759.0  469.53  4761.7  467.75  4783.2  465.70  4817.4  466.53
  4857.8  467.43  4879.3  465.73  4895.0  467.33  4981.1  467.17  4991.9  458.65
  4992.7  457.85  5000.8  458.65  5017.6  466.85  5125.3  466.77  5270.4  469.53
  5340.8  472.90  5362.5  476.68  5391.7  477.06  5406.6  479.57  5476.7  481.23
#Mann=5,-1,0
  4515.2    0.05       0  4524.6    0.16       0  4817.4    0.12       0
  4991.9    0.07       0  5000.8    0.12       0
Bank Sta=4759,5270.4
Exp/Cntr=0.3,0.1

Type RM Length L Ch R = 1,12457,465,465,465
BEGIN DESCRIPTION:
CHAFFIN CREEK 19.0
END DESCRIPTION:
XS GIS Cut Line= 3
      2837024.99      7081424.96      2836875.00      7080625.00
      2836524.99      7080324.99
#Sta/Elev= 30
  4216.9  490.21  4295.7  485.67  4348.3  481.46  4353.4  481.97  4389.8  480.89
  4476.2  476.26  4542.4  473.60  4573.8  471.79  4583.1  470.25  4627.5  468.03
  4633.1  467.87  4715.4  465.95  4894.3  466.52  4979.9  465.79  5000.1  458.18
  5000.9  457.38  5008.2  457.38  5009.0  458.18  5010.5  461.47  5020.6  466.09
  5080.7  465.63  5151.7  468.03  5251.6  474.42  5300.3  480.22  5314.5  483.30
  5335.4  486.26  5406.7  493.73  5433.7  495.16  5449.5  496.34  5491.8  497.12
#Mann=7,-1,0
  4216.9    0.05       0  4476.2    0.16       0  4633.1    0.12       0
  5000.1    0.07       0  5009.0    0.12       0  5251.6    0.16       0
  5433.7    0.12       0
Bank Sta=4627.5,5151.7
Exp/Cntr=0.3,0.1

Type RM Length L Ch R = 1,11992,634,634,634
BEGIN DESCRIPTION:
CHAFFIN CREEK 18.0
END DESCRIPTION:
XS GIS Cut Line= 3
      2837862.09      7081244.76      2837264.84      7080404.45
      2836752.04      7079908.97
#Sta/Elev= 30
  3969.2  487.85  4101.6  478.24  4196.5  472.10  4279.9  469.12  4488.8  466.14
  4633.1  465.86  4920.9  462.67  4962.7  465.17  4971.4  464.82  4977.5  463.02
  4986.1  458.05  4992.2  457.98  4993.0  457.18  5000.4  457.18  5001.3  457.98
  5003.3  457.98  5006.7  461.56  5013.8  464.36  5020.8  465.03  5063.3  463.54
  5160.0  466.14  5303.8  468.31  5336.2  469.69  5367.4  469.85  5438.1  473.12
  5483.2  473.89  5537.1  475.49  5558.2  474.63  5706.9  484.68  5713.2  484.83
#Mann=8,-1,0
  3969.2    0.12       0  4101.6    0.16       0  4279.9    0.12       0
  4992.2    0.07       0  5001.3    0.12       0  5336.2    0.16       0
  5483.2    0.05       0  5706.9    0.16       0
Bank Sta=4488.8,5160
Exp/Cntr=0.3,0.1

Type RM Length L Ch R = 1,11358,575,575,575
BEGIN DESCRIPTION:
CHAFFIN CREEK 17.0
END DESCRIPTION:
XS GIS Cut Line= 3
      2837875.95      7081095.39      2837775.00      7080175.00
      2837524.99      7079624.97
#Sta/Elev= 30
  4049.0  476.42  4270.7  470.18  4311.0  468.02  4441.7  467.01  4563.5  464.37
  4688.6  462.69  4689.0  462.68  4838.2  462.06  4904.5  460.87  4914.6  459.82
  4924.3  459.90  4929.3  461.26  4934.7  459.84  4944.7  459.70  4983.7  463.01
  4996.9  457.48  5002.2  456.96  5003.0  456.16  5011.4  456.96  5012.3  458.35
  5018.9  461.62  5029.8  463.19  5117.7  461.49  5229.6  464.37  5328.6  467.34
  5374.8  471.55  5437.6  481.09  5467.0  485.89  5541.7  495.17  5579.1  497.74
#Mann=6,-1,0
  4049.0    0.12       0  4688.6    0.05       0  4689.0    0.12       0
  5002.2    0.07       0  5011.4    0.12       0  5437.6    0.16       0
Bank Sta=4563.5,5229.6
Exp/Cntr=0.3,0.1

Type RM Length L Ch R = 1,10783,508,508,508
BEGIN DESCRIPTION:
CHAFFIN CREEK 16.0
END DESCRIPTION:
XS GIS Cut Line= 3
      2838803.02      7080605.82      2838278.73      7080025.98
      2837774.98      7079524.98
#Sta/Elev= 30
  4207.1  490.01  4220.7  488.92  4337.1  481.74  4362.0  481.93  4433.0  476.74
  4468.1  476.52  4489.7  474.03  4588.4  470.97  4734.7  463.10  4757.2  461.75
  4848.1  461.68  4901.2  461.30  4977.7  462.07  4982.8  459.42  4994.6  456.98
  4995.5  456.18  5003.9  456.98  5013.4  461.99  5020.5  462.12  5112.4  459.50
  5133.6  460.96  5381.1  460.83  5448.3  463.10  5497.0  466.83  5663.9  485.34
  5678.1  487.38  5685.1  490.09  5692.2  490.20  5695.7  493.50  5699.3  493.50
#Mann=10,-1,0
  4207.1    0.16       0  4220.7    0.12       0  4337.1    0.16       0
  4757.2    0.07       0  4848.1    0.12       0  4901.2    0.07       0
  4982.8    0.12       0  4994.6    0.07       0  5003.9    0.12       0
  5497.0    0.16       0
Bank Sta=4734.7,5448.3
Exp/Cntr=0.3,0.1

Type RM Length L Ch R = 1,10275,551,551,551
BEGIN DESCRIPTION:
CHAFFIN CREEK 15.0
END DESCRIPTION:
XS GIS Cut Line= 3
      2839174.97      7080474.96      2838625.00      7079675.00
      2838025.03      7078925.04
#Sta/Elev= 30
  4012.0  490.51  4034.3  486.39  4120.9  483.16  4285.3  467.40  4323.0  465.47
  4406.1  461.37  4485.5  460.86  4509.2  458.30  4903.6  461.74  4918.5  459.27
  4933.4  461.50  4960.4  461.47  4990.0  458.80  4999.7  456.10  5000.6  455.30
  5009.0  456.10  5010.8  460.73  5025.2  461.15  5153.3  460.42  5167.7  458.35
  5182.1  460.37  5225.3  458.59  5274.4  460.04  5316.9  461.37  5623.1  469.27
  5723.1  477.56  5851.2  493.29  5872.0  492.74  5900.8  497.12  5943.2  498.66
#Mann=5,-1,0
  4012.0    0.16       0  4323.0    0.12       0  4999.7    0.07       0
  5009.0    0.12       0  5274.4    0.05       0
Bank Sta=4406.1,5316.9
Exp/Cntr=0.3,0.1

Type RM Length L Ch R = 1,9724,358,358,358
BEGIN DESCRIPTION:
CHAFFIN CREEK 14.0
END DESCRIPTION:
XS GIS Cut Line= 3
      2839225.00      7080225.02      2839025.00      7079425.00
      2838674.98      7078874.96
#Sta/Elev= 30
  4192.7  473.91  4388.6  459.02  4424.4  458.20  4481.3  456.99  4499.4  455.28
  4512.3  456.44  4522.6  455.55  4540.6  456.80  4605.0  456.64  4628.2  457.80
  4751.9  458.09  4770.0  457.22  4852.4  458.81  4875.6  457.14  4904.0  458.63
  4980.0  458.75  4986.4  458.80  4994.6  454.28  4995.5  453.48  5003.9  454.28
  5007.0  458.52  5014.8  459.04  5313.7  455.84  5393.8  458.20  5437.3  461.03
  5506.4  469.75  5552.4  476.68  5574.4  478.49  5635.6  486.55  5669.3  490.20
#Mann=6,-1,0
  4192.7    0.12       0  4980.0    0.05       0  4994.6    0.03       0
  5003.9    0.05       0  5506.4    0.16       0  5635.6    0.05       0
Bank Sta=4424.4,5393.8
Exp/Cntr=0.3,0.1

Type RM Length L Ch R = 1,9366,349,349,349
BEGIN DESCRIPTION:
Mapping XS 5564b61e
END DESCRIPTION:
XS GIS Cut Line= 3
      2839670.21      7079750.79      2839321.26      7079313.30
      2838738.97      7078871.38
#Sta/Elev= 30
  4430.6  460.32  4472.7  459.67  4533.9  456.64  4609.0  453.68  4623.4  455.12
  4644.2  452.45  4658.7  455.23  4687.5  454.17  4693.9  455.96  4708.3  453.94
  4722.7  456.01  4788.6  456.27  4978.9  456.86  4990.2  456.56  4995.4  452.12
  4996.3  451.32  5004.7  452.12  5008.3  455.70  5014.6  456.57  5093.6  454.71
  5458.6  456.64  5463.8  458.30  5472.1  457.44  5488.7  458.66  5500.2  459.34
  5507.5  457.67  5513.7  460.22  5542.8  464.17  5712.8  482.48  5721.2  483.77
#Mann=7,-1,0
  4430.6    0.16       0  4472.7    0.12       0  4788.6    0.05       0
  4995.4    0.03       0  5004.7    0.05       0  5488.7    0.16       0
  5712.8    0.05       0
Bank Sta=4533.9,5458.6
Exp/Cntr=0.3,0.1

Type RM Length L Ch R = 1,9017,339,339,339
BEGIN DESCRIPTION:
double CHAFFIN CREEK 13.0
END DESCRIPTION:
XS GIS Cut Line= 3
      2841043.80      7079811.69      2839556.02      7079076.20
      2838805.32      7078552.27
#Sta/Elev= 30
  3257.1  489.52  3378.9  480.24  3501.2  474.73  3530.4  474.74  3536.0  476.86
  3561.8  474.66  3580.8  470.53  3597.7  471.48  3625.7  466.99  3670.6  467.47
  3687.4  464.19  3760.3  457.37  3768.9  458.44  3805.2  455.40  3927.2  453.29
  4024.0  450.68  4207.3  451.70  4267.8  451.44  4288.5  448.74  4289.4  447.94
  4297.8  448.74  4304.4  452.12  4377.1  452.02  4991.2  454.96  4997.4  450.92
  5012.2  454.83  5050.7  453.29  5515.5  455.47  5628.9  462.41  5832.2  484.86
#Mann=7,-1,0
  3257.1    0.05       0  3561.8    0.12       0  4207.3    0.05       0
  4267.8    0.07       0  4288.5    0.03       0  4297.8    0.07       0
  4377.1    0.05       0
Bank Sta=3927.2,5050.7
Exp/Cntr=0.3,0.1

Type RM Length L Ch R = 1,8678,918,918,918
BEGIN DESCRIPTION:
double CHAFFIN CREEK 12.0
END DESCRIPTION:
XS GIS Cut Line= 3
      2840836.87      7079396.62      2839625.00      7078725.00
      2838824.99      7078475.00
#Sta/Elev= 30
  3628.6  479.00  3669.4  477.12  3726.4  473.58  3769.0  469.23  3785.9  466.64
  3851.1  461.30  3867.2  458.66  3971.3  452.78  3986.0  452.67  4013.7  452.18
  4042.3  449.81  4110.9  450.80  4116.7  448.62  4122.4  449.13  4128.1  447.34
  4129.0  446.54  4137.4  447.34  4138.4  449.58  4145.2  450.80  4273.2  450.66
  4594.2  451.92  4911.2  452.52  4984.4  453.78  5000.4  451.25  5011.3  453.81
  5287.6  452.67  5533.3  455.28  5598.2  459.67  5733.4  473.96  5852.3  484.53
#Mann=8,-1,0
  3628.6    0.05       0  3669.4    0.12       0  3769.0    0.16       0
  3971.3    0.05       0  4128.1    0.03       0  4137.4    0.05       0
  4273.2    0.12       0  4594.2    0.05       0
Bank Sta=3986,5287.6
Exp/Cntr=0.3,0.1

Type RM Length L Ch R = 1,7760,458,458,458
BEGIN DESCRIPTION:
double CHAFFIN CREEK 11.0
END DESCRIPTION:
XS GIS Cut Line= 3
      2841040.04      7078625.82      2840258.76      7078198.72
      2839222.33      7077901.85
#Sta/Elev= 30
  4106.3  486.07  4118.1  483.39  4177.8  476.49  4362.8  458.56  4384.7  454.62
  4452.7  451.23  4477.6  449.21  4542.4  448.68  4706.3  449.23  4728.1  448.75
  4740.8  446.17  4745.3  445.66  4746.3  444.86  4755.2  445.66  4760.3  448.18
  4767.8  448.42  4972.8  450.43  5011.0  449.22  5027.5  450.38  5187.8  450.10
  5260.7  448.45  5298.3  449.81  5301.4  449.98  5648.6  451.23  5760.0  453.13
  5853.6  452.25  5939.1  456.42  6006.7  463.27  6011.9  462.44  6074.8  464.91
#Mann=8,-1,0
  4106.3    0.16       0  4542.4    0.12       0  4740.8    0.05       0
  4745.3    0.07       0  4755.2    0.05       0  4767.8    0.12       0
  5298.3    0.07       0  5301.4    0.05       0
Bank Sta=4452.7,5648.6
Exp/Cntr=0.3,0.1

Type RM Length L Ch R = 1,7302,927,927,927
BEGIN DESCRIPTION:
CHAFFIN CREEK 10.0
END DESCRIPTION:
XS GIS Cut Line= 3
      2841225.01      7077725.00      2840409.81      7077808.09
      2839474.96      7077524.99
#Sta/Elev= 30
  4186.3  487.70  4266.7  478.43  4276.8  473.11  4286.8  472.32  4301.5  473.99
  4338.2  469.37  4437.7  462.81  4608.5  457.18  4644.3  460.05  4719.1  460.48
  4744.1  458.45  4843.9  451.82  4861.6  450.95  4928.2  447.61  4970.3  448.20
  4980.4  446.75  4985.0  442.59  4985.7  441.79  4996.0  442.59  5005.6  447.21
  5021.2  448.11  5110.2  447.29  5125.7  446.00  5134.0  447.25  5374.9  449.02
  5725.1  447.90  5816.9  450.95  5862.0  455.15  5893.7  460.28  5982.5  469.56
#Mann=10,-1,0
  4186.3    0.05       0  4301.5    0.16       0  4644.3    0.12       0
  4744.1    0.07       0  4843.9    0.05       0  4928.2    0.12       0
  4985.0    0.07       0  4996.0    0.12       0  5110.2    0.05       0
  5893.7    0.16       0
Bank Sta=4861.6,5816.9
Exp/Cntr=0.3,0.1

Type RM Length L Ch R = 1,6375,800,800,800
BEGIN DESCRIPTION:
double CHAFFIN CREEK 9.0
END DESCRIPTION:
XS GIS Cut Line= 3
      2841224.96      7077574.98      2840675.00      7077325.00
      2840475.01      7076575.02
#Sta/Elev= 30
  4381.9  487.33  4502.7  477.59  4524.7  467.78  4534.5  466.79  4632.3  463.86
  4813.7  450.41  4890.1  446.89  4931.1  444.44  4971.7  446.31  4988.6  444.61
  4996.4  440.34  5003.5  446.70  5076.7  445.98  5152.6  445.87  5198.8  445.45
  5204.0  440.20  5224.0  445.79  5238.9  445.67  5244.7  444.72  5249.5  440.13
  5250.3  439.33  5260.6  440.13  5265.4  445.23  5348.6  450.41  5469.2  461.92
  5556.8  464.94  5638.0  469.98  5672.3  467.70  5675.4  467.81  5762.2  476.01
#Mann=9,-1,0
  4381.9    0.05       0  4890.1    0.12       0  5076.7    0.16       0
  5152.6    0.12       0  5249.5    0.07       0  5260.6    0.12       0
  5556.8    0.05       0  5672.3    0.16       0  5675.4    0.05       0
Bank Sta=4813.7,5348.6
Exp/Cntr=0.3,0.1

Type RM Length L Ch R = 1,5575,949,949,949
BEGIN DESCRIPTION:
CHAFFIN CREEK 8.0
END DESCRIPTION:
XS GIS Cut Line= 3
      2841461.48      7077293.78      2841061.46      7076843.75
      2840811.45      7076293.72
#Sta/Elev= 30
  4332.1  484.51  4364.2  482.07  4541.5  461.99  4652.1  451.28  4675.8  449.17
  4704.5  446.99  4732.1  446.31  4894.9  446.13  4938.0  445.42  4976.8  445.93
  4984.2  445.19  4989.7  442.35  4993.1  438.78  4993.8  437.98  5003.8  437.98
  5004.4  438.78  5013.3  449.17  5020.7  455.35  5042.7  460.58  5058.9  463.02
  5064.7  464.81  5075.6  466.78  5110.5  470.02  5124.8  472.06  5151.1  473.50
  5295.0  474.83  5387.5  474.19  5460.1  475.66  5496.1  477.79  5538.4  477.65
#Mann=7,-1,0
  4332.1    0.16       0  4652.1    0.05       0  4894.9    0.12       0
  4993.1    0.07       0  5004.4    0.12       0  5124.8    0.16       0
  5387.5    0.05       0
Bank Sta=4675.8,5013.3
Exp/Cntr=0.3,0.1

Type RM Length L Ch R = 1,4626,471,471,471
BEGIN DESCRIPTION:
CHAFFIN CREEK 7.0
END DESCRIPTION:
XS GIS Cut Line= 3
      2841783.33      7077147.92      2841733.33      7076397.92
      2841133.36      7076247.92
#Sta/Elev= 30
  4227.3  468.20  4270.3  464.51  4281.4  465.15  4340.5  463.17  4577.0  451.08
  4711.3  446.70  4758.4  446.27  4813.6  445.67  4841.6  446.58  4871.6  444.19
  4877.7  444.90  4891.7  443.11  4961.8  444.61  4971.9  442.89  4977.9  437.56
  5001.7  436.33  5002.3  435.53  5012.3  435.53  5013.0  436.33  5018.5  443.60
  5028.8  445.16  5082.2  443.95  5172.2  443.68  5248.5  446.27  5337.0  455.68
  5383.5  460.88  5419.6  466.35  5460.9  470.30  5554.5  473.77  5597.4  472.77
#Mann=6,-1,0
  4227.3    0.05       0  4813.6    0.12       0  5001.7    0.07       0
  5013.0    0.12       0  5082.2    0.05       0  5337.0    0.16       0
Bank Sta=4758.4,5248.5
Exp/Cntr=0.3,0.1

Type RM Length L Ch R = 1,4155,723,723,723
BEGIN DESCRIPTION:
CHAFFIN CREEK 6.0
END DESCRIPTION:
XS GIS Cut Line= 3
      2842711.89      7076516.43      2841975.00      7076125.00
      2841324.97      7075424.97
#Sta/Elev= 30
  4159.5  470.96  4195.1  469.64  4299.3  459.26  4393.8  452.88  4622.8  445.30
  4756.1  442.58  4858.8  442.86  4980.1  443.55  4991.1  437.02  4995.2  436.64
  4995.9  435.84  5006.7  436.64  5007.8  438.99  5015.2  443.57  5047.4  443.35
  5100.2  443.02  5121.2  441.00  5171.0  442.79  5213.0  442.13  5241.4  443.46
  5425.8  445.30  5503.3  447.49  5553.1  450.90  5682.7  456.33  5701.7  457.37
  5779.4  461.45  5842.9  467.00  5871.2  471.20  5899.6  471.68  5949.2  475.38
#Mann=7,-1,0
  4159.5    0.05       0  4858.8    0.12       0  4995.2    0.07       0
  5006.7    0.12       0  5047.4    0.05       0  5682.7    0.16       0
  5701.7    0.05       0
Bank Sta=4622.8,5425.8
Exp/Cntr=0.3,0.1

Type RM Length L Ch R = 1,3432,681,681,681
BEGIN DESCRIPTION:
CHAFFIN CREEK 5.0
END DESCRIPTION:
XS GIS Cut Line= 3
      2842925.00      7075675.00      2842325.00      7075575.00
      2841425.03      7075225.01
#Sta/Elev= 30
  4386.9  482.62  4468.0  479.67  4559.2  472.27  4579.5  468.55  4597.3  462.68
  4610.1  461.65  4663.2  458.29  4845.6  446.10  4925.6  443.46  4954.6  441.02
  4974.9  441.05  4985.0  438.94  4986.9  437.03  4987.5  436.23  4998.4  437.03
  5004.8  441.40  5010.1  441.75  5143.5  441.32  5166.8  440.01  5399.4  443.46
  5596.0  449.67  5707.6  451.05  5751.9  453.19  5782.6  455.12  5799.9  456.96
  5807.2  459.03  5837.1  460.91  5861.6  465.50  5883.0  466.94  5960.8  474.31
#Mann=8,-1,0
  4386.9    0.05       0  4610.1    0.16       0  4663.2    0.05       0
  4986.9    0.03       0  4998.4    0.05       0  5707.6    0.12       0
  5751.9    0.16       0  5883.0    0.05       0
Bank Sta=4925.6,5399.4
Exp/Cntr=0.3,0.1

Type RM Length L Ch R = 1,2751,698,698,698
BEGIN DESCRIPTION:
CHAFFIN CREEK 4.0
END DESCRIPTION:
XS GIS Cut Line= 3
      2843074.97      7075224.99      2842525.00      7074975.00
      2841624.97      7074424.98
#Sta/Elev= 30
  4392.6  479.50  4469.5  477.08  4572.6  467.67  4596.9  464.51  4634.2  462.48
  4741.6  452.27  4821.0  444.93  4872.1  441.97  4933.7  440.68  4974.7  440.82
  4982.2  435.83  4982.8  435.03  4993.7  435.83  4999.6  435.96  5004.4  440.54
  5017.7  440.99  5221.3  440.08  5242.8  437.59  5316.1  437.48  5324.9  437.53
  5331.5  440.06  5337.4  440.35  5374.1  438.70  5389.6  440.10  5564.8  441.97
  5738.0  447.06  5846.2  455.28  5906.3  459.34  5970.2  461.42  6051.5  467.43
#Mann=8,-1,0
  4392.6    0.05       0  4572.6    0.16       0  4741.6    0.05       0
  4933.7    0.16       0  4982.2    0.07       0  4993.7    0.16       0
  5017.7    0.05       0  5846.2    0.16       0
Bank Sta=4872.1,5564.8
Exp/Cntr=0.3,0.1
