HEC-RAS study ELM CREEK.prj: ELM CREEK Base Level Engineering

--- ELM CREEK.g01 (geometry) --- (continued)

Type RM Length L Ch R = 1,43809,770,770,770
BEGIN DESCRIPTION:
ELM CREEK 43.0
END DESCRIPTION:
XS GIS Cut Line= 3
      2830024.96      7062074.99      2829125.00      7061875.00
      2828575.01      7061575.01
#Sta/Elev= 30
  4064.0  471.58  4131.8  466.47  4136.9  467.96  4175.4  464.82  4364.9  458.19
  4432.7  453.99  4560.7  450.13  4641.5  447.63  4699.1  449.27  4760.5  448.97
  4777.2  447.67  4782.3  449.09  4801.5  449.21  4988.8  448.90  4994.0  446.88
  4999.7  440.54  5002.3  439.84  5002.8  439.04  5015.1  439.84  5037.6  449.27
  5081.3  448.01  5103.1  445.73  5119.3  447.39  5250.3  448.17  5310.0  450.13
  5397.4  454.99  5435.4  458.20  5517.0  468.20  5566.8  472.43  5612.4  474.05
#Mann=3,-1,0
  4064.0    0.05       0  5002.3    0.03       0  5015.1    0.05       0
Bank Sta=4560.7,5310
Exp/Cntr=0.3,0.1

Type RM Length L Ch R = 1,43039,1386,1386,1386
BEGIN DESCRIPTION:
ELM CREEK 42.0
END DESCRIPTION:
XS GIS Cut Line= 3
      2830175.00      7061875.00      2829525.00      7061525.00
      2828875.03      7061225.02
#Sta/Elev= 30
  4283.7  479.79  4483.3  466.93  4636.6  458.59  4772.1  454.03  4860.5  452.96
  4943.7  449.25  4964.3  448.76  4976.5  446.70  4986.3  439.67  4991.9  440.01
  4992.8  439.33  4993.3  438.53  5005.2  438.53  5005.7  439.33  5008.2  447.23
  5013.8  446.74  5019.1  447.66  5088.0  446.47  5173.8  447.54  5196.8  447.15
  5202.3  446.38  5231.2  447.36  5340.0  445.23  5374.4  446.33  5451.5  445.83
  5502.3  449.25  5528.6  450.55  5594.7  461.50  5631.8  465.98  5737.8  472.44
#Mann=3,-1,0
  4283.7    0.05       0  4992.8    0.03       0  5005.7    0.05       0
Bank Sta=4943.7,5502.3
Exp/Cntr=0.3,0.1

Type RM Length L Ch R = 1,41653,812,812,812
BEGIN DESCRIPTION:
ELM CREEK 41.0
END DESCRIPTION:
XS GIS Cut Line= 3
      2830524.95      7060924.99      2829625.00      7060775.00
      2829024.99      7060474.99
#Sta/Elev= 30
  4096.3  473.13  4167.2  467.98  4339.2  449.33  4423.5  447.49  4684.3  444.06
  4785.6  445.31  4872.2  444.93  4980.8  446.27  4988.4  444.45  4998.5  439.32
  4999.7  437.07  5000.2  436.27  5012.1  436.27  5012.6  437.07  5017.1  438.79
  5022.6  437.11  5031.0  439.49  5039.4  445.54  5045.0  444.56  5053.4  446.30
  5179.2  444.47  5268.6  445.36  5313.3  446.94  5344.1  446.52  5362.4  447.49
  5447.5  449.03  5499.3  451.88  5545.3  455.14  5620.8  464.37  5679.5  470.21
#Mann=6,-1,0
  4096.3    0.16       0  4339.2    0.05       0  4872.2    0.12       0
  4999.7    0.07       0  5012.6    0.12       0  5499.3    0.05       0
Bank Sta=4423.5,5362.4
Exp/Cntr=0.3,0.1

Type RM Length L Ch R = 1,40841,661,661,661
BEGIN DESCRIPTION:
ELM CREEK 40.0
END DESCRIPTION:
XS GIS Cut Line= 3
      2830625.03      7060925.03      2829875.00      7060225.00
      2829325.00      7059975.00
#Sta/Elev= 30
  3987.5  480.18  4136.3  465.21  4192.7  457.95  4317.2  446.84  4395.4  444.64
  4589.2  443.24  4603.1  441.16  4617.0  441.02  4624.3  441.23  4638.5  443.62
  4857.9  443.34  4886.2  442.33  4958.1  444.27  4978.0  444.73  4985.4  443.52
  4993.1  436.46  4993.6  435.66  5005.5  435.66  5006.0  436.46  5010.0  437.72
  5016.2  437.72  5027.7  445.03  5125.5  443.54  5203.6  446.02  5216.9  446.84
  5292.5  451.72  5384.7  461.18  5459.4  467.70  5464.9  467.07  5617.6  470.39
#Mann=6,-1,0
  3987.5    0.16       0  4395.4    0.05       0  4958.1    0.12       0
  4993.1    0.07       0  5006.0    0.12       0  5203.6    0.16       0
Bank Sta=4317.2,5216.9
Exp/Cntr=0.3,0.1

Type RM Length L Ch R = 1,40180,799,799,799
BEGIN DESCRIPTION:
ELM CREEK 39.0
END DESCRIPTION:
XS GIS Cut Line= 3
      2830924.96      7060274.97      2830025.00      7059625.00
      2829425.01      7059725.00
#Sta/Elev= 30
  3890.7  464.55  3998.6  453.06  4069.8  448.39  4120.6  446.38  4141.2  446.56
  4185.0  444.52  4321.2  441.96  4786.2  441.89  4907.6  442.48  4972.6  444.52
  4978.8  444.06  4991.3  435.98  4991.8  435.18  5003.8  435.18  5004.3  435.98
  5011.0  442.74  5118.7  446.13  5125.0  446.38  5150.4  448.11  5155.4  447.54
  5193.5  451.07  5211.2  454.07  5216.3  453.58  5244.1  457.33  5254.3  457.64
  5272.0  460.50  5277.1  460.05  5322.7  464.12  5393.7  468.25  5609.1  470.46
#Mann=6,-1,0
  3890.7    0.16       0  4141.2    0.12       0  4991.3    0.07       0
  5004.3    0.12       0  5118.7    0.16       0  5322.7    0.12       0
Bank Sta=4120.6,5125
Exp/Cntr=0.3,0.1

Type RM Length L Ch R = 1,39381,1244,1244,1244
BEGIN DESCRIPTION:
ELM CREEK 38.0
END DESCRIPTION:
XS GIS Cut Line= 3
      2831175.04      7059324.99      2830575.00      7059425.00
      2829775.04      7059225.01
#Sta/Elev= 30
  4405.1  471.60  4433.0  466.02  4438.1  468.71  4490.1  454.31  4493.8  452.90
  4498.9  454.71  4516.7  449.33  4536.9  446.21  4598.6  445.29  4600.1  445.26
  4729.6  444.28  4841.1  440.01  4871.5  441.45  4891.8  434.89  4905.5  434.79
  4906.0  433.99  4918.5  434.79  4932.3  440.30  4972.9  442.79  4980.5  435.28
  4993.1  434.80  5003.3  435.60  5010.9  442.81  5085.6  441.57  5237.6  443.29
  5415.4  441.90  5522.9  445.29  5547.3  447.18  5773.6  465.76  5838.0  468.26
#Mann=6,-1,0
  4405.1    0.12       0  4490.1    0.07       0  4600.1    0.12       0
  4905.5    0.07       0  4918.5    0.12       0  5547.3    0.16       0
Bank Sta=4598.6,5522.9
Exp/Cntr=0.3,0.1

Type RM Length L Ch R = 1,38137,600,600,600
BEGIN DESCRIPTION:
ELM CREEK 37.0
END DESCRIPTION:
XS GIS Cut Line= 3
      2831574.97      7058824.99      2830966.89      7058606.31
      2829850.19      7058840.04
#Sta/Elev= 30
  4385.3  475.64  4431.3  471.96  4487.5  464.30  4548.9  458.20  4555.3  456.66
  4635.7  445.98  4712.7  442.12  4772.1  439.99  4895.4  439.10  4969.8  440.26
  4980.4  438.26  4987.1  432.86  4987.7  432.06  4999.7  432.06  5000.3  432.86
  5001.6  435.47  5012.3  440.45  5019.1  440.62  5227.6  438.52  5243.8  439.45
  5319.5  440.01  5380.8  439.02  5401.2  439.92  5855.3  442.12  5942.5  445.24
  6034.7  453.47  6055.1  453.52  6096.0  458.49  6122.5  458.90  6172.4  463.27
#Mann=5,-1,0
  4385.3    0.05       0  4772.1    0.12       0  4987.1    0.07       0
  5000.3    0.12       0  5942.5    0.16       0
Bank Sta=4712.7,5855.3
Exp/Cntr=0.3,0.1

Type RM Length L Ch R = 1,37537,868,868,868
BEGIN DESCRIPTION:
ELM CREEK 36.0
END DESCRIPTION:
XS GIS Cut Line= 3
      2831624.97      7058674.97      2831025.00      7058175.00
      2829924.96      7057774.98
#Sta/Elev= 30
  4205.2  477.65  4276.1  474.35  4325.6  469.99  4382.8  462.03  4489.6  451.94
  4588.5  447.30  4602.8  445.31  4733.2  442.04  4787.5  441.04  4859.7  439.18
  4979.0  438.66  4982.9  436.61  4988.8  436.61  4989.6  429.82  4990.2  429.02
  5002.8  429.82  5018.1  430.13  5026.8  438.43  5032.1  435.68  5039.4  438.58
  5118.5  438.67  5260.8  437.77  5299.7  434.72  5337.3  437.59  5404.2  438.04
  5688.5  439.16  5750.9  441.04  5820.8  445.47  6080.2  470.88  6156.7  474.14
#Mann=7,-1,0
  4205.2    0.05       0  4733.2    0.07       0  4859.7    0.12       0
  4989.6    0.07       0  5002.8    0.12       0  5299.7    0.16       0
  5404.2    0.05       0
Bank Sta=4787.5,5750.9
Exp/Cntr=0.3,0.1

Type RM Length L Ch R = 1,36669,256,256,256
BEGIN DESCRIPTION:
Mapping XS c8883421
END DESCRIPTION:
XS GIS Cut Line= 3
      2832069.32      7057703.53      2831687.38      7057356.31
      2830308.54      7057304.28
#Sta/Elev= 30
  3930.8  466.24  4024.9  463.44  4173.5  455.91  4272.9  449.00  4348.9  446.05
  4496.2  440.01  4509.4  437.31  4549.4  439.00  4649.5  436.23  4693.8  433.63
  4719.6  433.63  4739.6  436.19  4792.9  436.65  4929.7  435.90  4979.7  437.04
  4989.7  428.08  4992.8  427.01  4993.7  426.21  5006.8  427.01  5019.8  435.43
  5090.0  436.73  5189.1  437.01  5321.1  436.72  5400.0  437.47  5469.9  440.01
  5570.2  447.62  5670.2  457.73  5680.2  460.29  5720.3  462.32  5826.8  463.05
#Mann=9,-1,0
  3930.8    0.05       0  4348.9    0.16       0  4693.8    0.12       0
  4792.9    0.16       0  4992.8    0.07       0  5006.8    0.16       0
  5090.0    0.12       0  5189.1    0.16       0  5321.1    0.05       0
Bank Sta=4496.2,5469.9
Exp/Cntr=0.3,0.1

Type RM Length L Ch R = 1,36413,796,796,796
BEGIN DESCRIPTION:
Mapping XS ad8799d9
END DESCRIPTION:
XS GIS Cut Line= 3
      2832269.01      7057217.43      2831253.35      7057121.94
      2830386.55      7057069.93
#Sta/Elev= 30
  3952.6  464.76  4032.0  464.31  4067.1  456.35  4117.3  454.47  4140.6  458.10
  4157.5  453.28  4277.3  446.42  4452.7  439.71  4581.1  436.96  4830.5  437.26
  4860.6  436.65  4880.7  431.52  4961.0  436.84  4969.4  430.82  4984.1  427.12
  4985.0  426.32  4998.1  427.12  5005.6  429.94  5011.2  436.47  5031.2  433.04
  5101.3  439.45  5151.4  432.14  5201.5  440.46  5231.6  437.29  5312.8  439.71
  5492.0  448.98  5572.8  460.01  5671.9  468.08  5722.4  473.26  5841.1  477.10
#Mann=7,-1,0
  3952.6    0.08       0  4277.3    0.05       0  4581.1    0.12       0
  4984.1    0.07       0  4998.1    0.12       0  5572.8    0.16       0
  5671.9    0.05       0
Bank Sta=4452.7,5312.8
Exp/Cntr=0.3,0.1

Type RM Length L Ch R = 1,35617,659,659,659
BEGIN DESCRIPTION:
Mapping XS 95f2342b
END DESCRIPTION:
XS GIS Cut Line= 3
      2832199.54      7056818.12      2831626.62      7056583.74
      2830784.63      7056557.70
#Sta/Elev= 30
  4349.6  462.32  4453.7  455.63  4507.1  454.74  4555.2  448.82  4560.6  449.86
  4685.6  438.11  4691.1  437.99  4744.8  436.21  4775.9  432.42  4792.9  434.27
  4830.4  433.02  4840.7  432.10  4862.3  434.89  4953.1  434.67  4980.2  425.85
  4993.2  425.44  4994.1  424.64  5007.2  425.44  5020.3  434.23  5030.3  435.14
  5214.8  438.11  5320.4  440.52  5430.4  446.48  5450.5  442.31  5510.5  451.75
  5540.5  452.22  5580.5  461.23  5631.8  460.46  5680.6  461.11  5811.0  469.63
#Mann=6,-1,0
  4349.6    0.05       0  4691.1    0.16       0  4830.4    0.12       0
  4993.2    0.07       0  5007.2    0.12       0  5631.8    0.16       0
Bank Sta=4685.6,5214.8
Exp/Cntr=0.3,0.1

Type RM Length L Ch R = 1,34958,792,792,792
BEGIN DESCRIPTION:
ELM CREEK 33.0
END DESCRIPTION:
XS GIS Cut Line= 3
      2832578.94      7056278.24      2831575.00      7055925.00
      2830874.98      7056025.00
#Sta/Elev= 30
  3957.4  463.52  4025.2  462.13  4098.4  457.37  4194.5  458.24  4205.4  458.64
  4222.3  450.95  4284.2  449.85  4331.6  445.85  4371.8  440.97  4469.4  436.31
  4614.2  432.08  4661.2  433.28  4682.4  430.79  4732.8  433.82  4794.7  432.39
  4980.5  434.61  4989.9  426.22  4993.4  425.34  4994.4  424.54  5007.5  425.34
  5011.5  431.16  5019.0  434.14  5102.5  432.81  5211.9  435.55  5237.0  436.31
  5314.6  439.49  5597.5  469.02  5668.2  474.13  5717.1  474.35  5728.8  474.54
#Mann=7,-1,0
  3957.4    0.05       0  4194.5    0.16       0  4331.6    0.12       0
  4993.4    0.07       0  5007.5    0.12       0  5211.9    0.16       0
  5717.1    0.05       0
Bank Sta=4469.4,5237
Exp/Cntr=0.3,0.1

Type RM Length L Ch R = 1,34166,820,820,820
BEGIN DESCRIPTION:
ELM CREEK 32.0
END DESCRIPTION:
XS GIS Cut Line= 3
      2832425.00      7055675.00      2831825.00      7055175.00
      2830925.01      7055475.00
#Sta/Elev= 30
  4197.5  463.34  4289.3  458.51  4332.2  453.62  4340.0  451.56  4376.2  448.28
  4408.4  444.40  4418.1  442.60  4488.4  437.21  4544.2  434.56  4644.6  430.87
  4730.6  430.16  4800.8  431.91  4872.4  429.88  4878.9  431.14  4964.9  432.80
  4971.4  431.16  4975.3  425.97  4992.6  425.24  4993.5  424.44  5006.7  425.24
  5020.7  432.25  5031.2  433.21  5078.1  432.57  5210.4  431.69  5373.6  434.56
  5463.4  435.96  5589.9  440.48  5750.7  457.79  5790.2  462.16  5927.2  470.10
#Mann=7,-1,0
  4197.5    0.05       0  4376.2    0.16       0  4408.4    0.12       0
  4992.6    0.07       0  5006.7    0.12       0  5078.1    0.05       0
  5750.7    0.16       0
Bank Sta=4544.2,5373.6
Exp/Cntr=0.3,0.1

Type RM Length L Ch R = 1,33346,883,883,883
BEGIN DESCRIPTION:
ELM CREEK 31.0
END DESCRIPTION:
XS GIS Cut Line= 3
      2832838.93      7055088.93      2832275.00      7054525.00
      2831374.99      7054024.99
#Sta/Elev= 30
  4181.5  461.70  4229.5  462.40  4271.9  461.41  4328.5  459.35  4469.9  451.65
  4663.1  432.64  4700.6  430.69  4752.7  429.71  4908.3  430.81  4964.9  432.14
  4981.9  430.92  4987.0  425.74  4994.8  425.60  4995.8  424.80  5008.0  424.80
  5009.0  425.60  5014.5  430.73  5024.8  432.05  5056.2  431.19  5390.8  429.82
  5485.8  432.29  5523.5  431.51  5587.8  432.64  5676.8  435.51  5713.4  437.96
  5734.6  440.86  5848.4  453.35  5891.9  459.26  5958.3  464.44  6008.6  467.41
#Mann=7,-1,0
  4181.5    0.05       0  4700.6    0.12       0  4994.8    0.07       0
  5009.0    0.12       0  5056.2    0.05       0  5734.6    0.16       0
  5958.3    0.05       0
Bank Sta=4663.1,5587.8
Exp/Cntr=0.3,0.1

Type RM Length L Ch R = 1,32463,645,645,645
BEGIN DESCRIPTION:
ELM CREEK 30.0
END DESCRIPTION:
XS GIS Cut Line= 3
      2833187.74      7054449.38      2832525.00      7053775.00
      2831424.96      7053875.00
#Sta/Elev= 30
  4068.8  447.73  4092.7  446.72  4099.5  446.38  4151.6  444.39  4201.1  440.03
  4243.5  434.63  4292.7  432.10  4338.1  430.97  4450.2  429.14  4833.9  428.91
  4929.5  429.14  4972.0  430.64  4986.0  424.01  4987.0  423.21  5000.2  424.01
  5007.2  429.35  5010.8  430.27  5094.9  429.24  5225.2  427.92  5335.6  429.18
  5536.5  428.41  5623.1  429.86  5687.4  432.10  5757.4  434.29  5821.8  438.17
  5888.3  444.67  5919.7  447.66  5931.4  448.81  6068.7  463.24  6118.9  466.63
#Mann=14,-1,0
  4068.8    0.12       0  4092.7    0.05       0  4099.5    0.12       0
  4338.1    0.16       0  4450.2    0.05       0  4833.9    0.16       0
  4986.0    0.07       0  5000.2    0.16       0  5094.9    0.05       0
  5623.1    0.12       0  5821.8    0.16       0  5888.3    0.12       0
  5919.7    0.16       0  5931.4    0.05       0
Bank Sta=4292.7,5687.4
Exp/Cntr=0.3,0.1

Type RM Length L Ch R = 1,31818,1007,1007,1007
BEGIN DESCRIPTION:
double ELM CREEK 29.0
END DESCRIPTION:
XS GIS Cut Line= 3
      2833507.21      7053039.64      2832896.07      7053199.38
      2831805.75      7053004.92
#Sta/Elev= 30
  4119.0  451.51  4206.7  442.40  4372.2  431.83  4472.6  428.39  4507.7  429.59
  4558.0  428.97  4593.3  430.21  4782.2  430.63  4792.4  429.10  4798.7  422.61
  4799.7  421.81  4813.0  422.61  4822.9  429.44  4833.0  430.60  4944.8  428.58
  4977.6  429.30  4985.4  428.28  4995.5  423.19  5017.8  429.51  5122.5  427.79
  5149.4  426.11  5188.5  426.47  5208.9  427.98  5249.5  426.18  5269.8  428.28
  5316.1  430.16  5493.3  428.84  5633.1  431.83  5706.6  436.13  5858.2  452.40
#Mann=8,-1,0
  4119.0    0.16       0  4206.7    0.12       0  4472.6    0.16       0
  4507.7    0.12       0  4798.7    0.07       0  4813.0    0.12       0
  5017.8    0.07       0  5122.5    0.05       0
Bank Sta=4372.2,5633.1
Exp/Cntr=0.3,0.1

Type RM Length L Ch R = 1,30811,884,884,884
BEGIN DESCRIPTION:
ELM CREEK 28.0
END DESCRIPTION:
XS GIS Cut Line= 3
      2833324.97      7052624.98      2832725.00      7052225.00
      2832024.98      7052225.00
#Sta/Elev= 30
  4273.3  455.86  4381.4  454.98  4477.3  444.98  4496.6  442.07  4613.8  431.10
  4619.5  430.50  4647.3  427.84  4669.9  427.59  4683.4  423.65  4692.4  422.45
  4713.4  427.21  4778.0  427.81  4863.7  426.26  4893.7  427.77  4958.3  428.31
  4971.8  425.75  4980.9  421.36  4982.3  418.65  4984.8  417.85  5000.5  418.65
  5004.4  421.54  5024.4  428.55  5204.4  426.92  5311.7  429.88  5323.6  430.50
  5414.4  435.52  5524.4  447.24  5544.4  447.63  5634.4  456.10  5694.4  458.33
#Mann=7,-1,0
  4273.3    0.16       0  4477.3    0.05       0  4496.6    0.16       0
  4613.8    0.12       0  4982.3    0.07       0  5000.5    0.12       0
  5311.7    0.05       0
Bank Sta=4619.5,5323.6
Exp/Cntr=0.3,0.1

Type RM Length L Ch R = 1,29927,718,718,718
BEGIN DESCRIPTION:
ELM CREEK 27.0
END DESCRIPTION:
XS GIS Cut Line= 3
      2833775.01      7052325.01      2832975.00      7051525.00
      2832274.99      7051525.00
#Sta/Elev= 30
  3872.8  463.75  3930.8  461.32  3971.8  458.19  4028.4  450.34  4113.2  442.01
  4198.1  435.60  4387.8  428.80  4579.9  424.47  4594.1  426.06  4608.2  424.38
  4687.2  425.07  4707.2  425.87  4844.6  424.59  4882.6  426.33  4975.9  427.12
  4991.6  418.37  4994.1  417.57  5009.8  418.37  5024.2  424.87  5034.2  426.29
  5254.2  426.66  5288.0  428.80  5374.2  437.04  5407.4  441.90  5411.4  442.26
  5474.2  447.53  5514.2  452.55  5574.2  456.92  5614.2  458.34  5704.2  457.74
#Mann=10,-1,0
  3872.8    0.05       0  3930.8    0.16       0  4198.1    0.05       0
  4687.2    0.12       0  4844.6    0.16       0  4882.6    0.12       0
  4991.6    0.07       0  5009.8    0.12       0  5407.4    0.07       0
  5411.4    0.05       0
Bank Sta=4387.8,5288
Exp/Cntr=0.3,0.1

Type RM Length L Ch R = 1,29209,331,331,331
BEGIN DESCRIPTION:
Mapping XS 4de2c635
END DESCRIPTION:
XS GIS Cut Line= 3
      2834265.53      7051609.80      2833640.50      7051271.24
      2832503.35      7051201.80
#Sta/Elev= 30
  3955.7  453.03  4100.4  449.76  4182.1  443.45  4217.9  437.98  4275.3  431.82
  4368.5  427.38  4615.9  423.48  4672.0  424.90  4841.9  425.33  4982.6  425.59
  4992.6  422.87  4993.6  417.14  4996.1  416.34  5011.8  417.14  5016.4  417.35
  5022.7  423.09  5032.7  425.94  5062.8  424.28  5082.8  425.37  5139.2  425.27
  5173.0  424.38  5238.3  426.96  5303.2  426.63  5403.4  429.16  5483.5  426.71
  5525.8  427.38  5565.6  429.00  5605.3  430.90  5733.8  441.48  5805.8  446.96
#Mann=9,-1,0
  3955.7    0.05       0  4841.9    0.12       0  4993.6    0.07       0
  5011.8    0.12       0  5139.2    0.16       0  5238.3    0.12       0
  5565.6    0.07       0  5605.3    0.12       0  5733.8    0.05       0
Bank Sta=4368.5,5525.8
Exp/Cntr=0.3,0.1

Type RM Length L Ch R = 1,28878,636,636,636
BEGIN DESCRIPTION:
ELM CREEK 26.0
END DESCRIPTION:
XS GIS Cut Line= 3
      2834456.47      7051054.23      2833423.49      7051002.15
      2832486.03      7050967.42
#Sta/Elev= 30
  3966.2  448.81  4007.7  447.28  4107.9  434.28  4160.0  431.25  4245.9  427.89
  4407.0  426.43  4508.4  425.82  4578.4  423.98  4728.6  424.23  4758.7  423.09
  4952.5  425.04  4968.9  425.54  4979.0  419.83  4979.9  418.13  4982.4  417.33
  4995.6  417.33  4998.1  418.13  5000.5  418.21  5009.0  424.91  5051.5  425.34
  5150.6  423.65  5219.1  426.35  5327.6  426.43  5439.3  427.36  5569.4  429.93
  5669.4  433.22  5729.5  437.79  5769.5  442.53  5879.6  453.17  5938.6  456.36
#Mann=7,-1,0
  3966.2     0.1       0  4160.0    0.05       0  4952.5    0.12       0
  4979.9    0.07       0  4998.1    0.12       0  5051.5    0.07       0
  5150.6    0.05       0
Bank Sta=4407,5327.6
Exp/Cntr=0.3,0.1

Type RM Length L Ch R = 1,28242,342,342,342
BEGIN DESCRIPTION:
ELM CREEK 25.0
END DESCRIPTION:
XS GIS Cut Line= 3
      2834875.05      7050875.02      2833475.00      7050375.00
      2832774.96      7050274.99
#Sta/Elev= 30
  3504.2  461.29  3929.0  440.56  3965.6  437.39  4052.7  434.68  4204.7  425.56
  4473.2  423.31  4498.7  421.11  4529.5  423.85  4591.1  420.25  4608.6  421.96
  4647.3  421.44  4652.7  423.05  4757.2  421.86  4770.5  423.75  4789.1  422.21
  4801.3  418.74  4821.0  422.26  4969.6  424.09  4975.5  421.00  4979.1  416.79
  4981.6  415.99  4997.3  416.79  5001.0  420.38  5011.1  423.95  5113.8  425.56
  5354.5  441.32  5384.8  446.02  5475.7  453.27  5596.9  457.29  5698.0  457.98
#Mann=3,-1,0
  3504.2    0.05       0  4979.1    0.03       0  4997.3    0.05       0
Bank Sta=4204.7,5113.8
Exp/Cntr=0.3,0.1

Type RM Length L Ch R = 1,27900,524,524,524
BEGIN DESCRIPTION:
Mapping XS b643f5e1
END DESCRIPTION:
XS GIS Cut Line= 3
      2835003.31      7050125.41      2833492.93      7050038.60
      2832920.01      7050151.45
#Sta/Elev= 30
  3511.4  448.09  3569.8  443.65  3599.9  443.30  3605.2  441.87  3610.3  443.16
  3629.9  439.32  3720.1  440.33  3870.3  433.66  3966.2  432.44  4150.9  426.37
  4178.8  425.32  4391.2  422.12  4411.2  420.04  4441.2  422.88  4527.7  422.63
  4642.2  421.68  4661.6  418.51  4681.6  418.23  4731.7  422.25  4924.0  423.47
  4972.1  423.75  4989.4  415.62  4991.9  414.82  5007.6  415.62  5012.2  423.35
  5043.6  424.92  5058.2  425.32  5256.6  435.44  5496.6  455.28  5608.2  457.85
#Mann=9,-1,0
  3511.4    0.05       0  3966.2     0.1       0  4150.9    0.05       0
  4527.7    0.12       0  4642.2    0.05       0  4924.0    0.16       0
  4989.4    0.07       0  5007.6    0.16       0  5043.6    0.05       0
Bank Sta=4178.8,5058.2
Exp/Cntr=0.3,0.1

Type RM Length L Ch R = 1,27376,497,497,497
BEGIN DESCRIPTION:
Mapping XS ee8f9a58
END DESCRIPTION:
XS GIS Cut Line= 3
      2835164.54      7049931.84      2833495.32      7049542.45
      2832831.12      7049948.85
#Sta/Elev= 30
  3208.2  457.52  3361.8  450.12  3556.9  444.33  3703.1  436.74  3803.3  428.98
  3985.9  424.35  4293.5  421.72  4405.8  420.21  4419.4  415.90  4420.6  413.42
  4423.1  412.62  4438.8  413.42  4439.9  415.65  4446.9  419.50  4460.5  418.80
  4481.0  422.51  4674.5  422.04  4969.3  422.95  4981.2  416.90  4996.5  414.03
  5011.9  414.68  5015.6  417.59  5025.2  420.82  5039.8  422.85  5102.6  424.35
  5128.0  428.07  5246.6  433.59  5507.2  444.97  5607.9  452.03  5700.9  454.53
#Mann=9,-1,0
  3208.2    0.05       0  4293.5    0.16       0  4405.8    0.12       0
  4420.6    0.07       0  4438.8    0.12       0  4674.5    0.16       0
  5015.6    0.12       0  5025.2    0.16       0  5246.6    0.05       0
Bank Sta=3985.9,5102.6
Exp/Cntr=0.3,0.1

Type RM Length L Ch R = 1,26879,656,656,656
BEGIN DESCRIPTION:
double ELM CREEK 24.0
END DESCRIPTION:
XS GIS Cut Line= 3
      2834560.31      7048133.22      2833154.02      7049316.91
      2832535.98      7049816.90
#Sta/Elev= 30
  3124.3  450.64  3150.7  451.67  3165.7  453.90  3298.4  449.66  3446.2  441.35
  3519.9  443.00  3696.8  432.22  3782.6  435.64  3966.2  423.64  4480.7  420.90
  4486.5  420.91  4520.1  419.78  4525.3  412.89  4527.8  412.09  4543.5  412.89
  4548.7  420.35  4618.5  420.41  4625.5  420.21  4776.3  421.05  4882.7  421.47
  4979.4  420.44  5010.6  413.92  5025.0  421.94  5080.9  422.74  5097.6  423.64
  5225.5  433.03  5376.7  444.72  5403.5  446.28  5487.1  452.49  5757.4  454.43
#Mann=18,-1,0
  3124.3    0.16       0  3150.7    0.12       0  3165.7     0.1       0
  3298.4    0.08       0  3446.2    0.05       0  4480.7    0.16       0
  4486.5    0.05       0  4525.3    0.07       0  4543.5    0.05       0
  4618.5    0.07       0  4625.5    0.16       0  4776.3    0.12       0
  4882.7    0.16       0  4979.4    0.12       0  5080.9    0.16       0
  5225.5    0.12       0  5376.7    0.16       0  5403.5    0.05       0
Bank Sta=3966.2,5097.6
Exp/Cntr=0.3,0.1

Type RM Length L Ch R = 1,26223,703,703,703
BEGIN DESCRIPTION:
double ELM CREEK 23.0
END DESCRIPTION:
XS GIS Cut Line= 3
      2833935.25      7048323.86      2832900.54      7048747.47
      2832226.94      7049528.71
#Sta/Elev= 30
  3830.9  444.88  4293.1  426.36  4351.9  427.32  4484.3  422.28  4591.8  419.52
  4643.0  418.91  4674.0  412.42  4691.0  420.20  4764.5  419.11  4765.9  419.15
  4922.0  419.17  4986.2  420.64  4999.0  412.10  5001.5  411.30  5017.2  412.10
  5022.3  418.31  5036.6  420.09  5305.4  420.44  5327.3  418.47  5341.4  420.65
  5379.2  422.28  5440.3  424.50  5454.6  422.93  5518.2  429.87  5567.6  432.23
  5575.3  430.86  5596.1  433.99  5667.8  437.13  5872.6  448.65  5980.5  452.31
#Mann=9,-1,0
  3830.9    0.05       0  4591.8    0.16       0  4764.5    0.12       0
  4765.9    0.16       0  4922.0    0.12       0  4999.0    0.07       0
  5017.2    0.12       0  5341.4    0.16       0  5667.8    0.05       0
Bank Sta=4484.3,5379.2
Exp/Cntr=0.3,0.1

Type RM Length L Ch R = 1,25520,177,177,177
BEGIN DESCRIPTION:
Mapping XS d40db136
END DESCRIPTION:
XS GIS Cut Line= 3
      2833935.62      7048285.13      2832538.07      7048233.05
      2830949.78      7048215.69
#Sta/Elev= 30
  3714.4  444.70  3916.7  437.20  4015.7  433.25  4215.4  432.52  4545.8  420.78
  4705.7  418.44  4889.0  419.57  4965.9  419.80  4975.9  417.55  4986.7  412.09
  4989.2  411.29  5005.1  412.09  5015.9  412.81  5035.9  418.83  5045.9  419.56
  5115.2  419.14  5286.0  417.23  5316.0  418.70  5482.6  417.60  5946.0  420.08
  5966.0  418.08  5986.0  420.13  6095.5  420.65  6106.0  417.63  6123.0  420.78
  6416.1  424.16  6566.1  430.36  6590.7  432.43  6616.1  434.48  6701.3  436.64
#Mann=10,-1,0
  3714.4    0.05       0  3916.7    0.08       0  4015.7    0.05       0
  4889.0    0.12       0  4986.7    0.07       0  5005.1    0.12       0
  5115.2    0.16       0  5482.6    0.05       0  6095.5    0.08       0
  6590.7    0.05       0
Bank Sta=4545.8,6123
Exp/Cntr=0.3,0.1

Type RM Length L Ch R = 1,25343,856,856,856
BEGIN DESCRIPTION:
Mapping XS 2363d6d6
END DESCRIPTION:
XS GIS Cut Line= 4
      2834005.11      7048172.29      2832598.84      7048102.84
      2832104.05      7048085.48      2831028.86      7048007.44
#Sta/Elev= 30
  3549.3  446.85  3839.8  437.06  3917.6  436.94  4003.1  439.74  4060.0  438.89
  4406.0  422.91  4532.9  420.43  4760.9  419.06  4790.9  416.20  4814.0  418.52
  4971.1  419.29  5001.2  413.05  5007.2  414.27  5021.2  419.01  5106.2  418.61
  5201.3  417.43  5271.3  419.85  5301.3  417.85  5361.4  418.15  5381.4  415.10
  5382.2  411.74  5384.7  410.94  5400.6  411.74  5401.4  417.82  5403.4  417.95
  5502.4  417.83  5945.1  418.23  6147.3  420.43  6383.9  427.96  6530.4  443.66
#Mann=8,-1,0
  3549.3    0.16       0  3917.6    0.05       0  5007.2    0.16       0
  5106.2    0.12       0  5382.2    0.03       0  5400.6    0.12       0
  5403.4     0.1       0  5502.4    0.05       0
Bank Sta=4532.9,6147.3
Exp/Cntr=0.3,0.1

Type RM Length L Ch R = 1,24487,576,576,576
BEGIN DESCRIPTION:
Mapping XS 3822386e
END DESCRIPTION:
XS GIS Cut Line= 3
      2832729.02      7047425.77      2831982.52      7047764.30
      2831045.06      7047781.66
#Sta/Elev= 30
  4158.1  444.25  4260.5  441.24  4381.5  434.77  4456.2  430.18  4559.5  421.17
  4616.2  418.63  4634.7  416.87  4667.6  415.78  4675.0  412.05  4689.6  411.17
  4704.4  416.30  4772.8  417.30  4801.4  415.88  4832.3  417.12  4963.0  418.49
  4977.8  417.77  4985.3  414.10  4986.1  409.70  4988.6  408.90  5004.6  409.70
  5015.3  417.69  5025.3  418.46  5175.3  415.60  5365.4  418.08  5405.4  417.40
  5560.3  418.63  5695.4  423.04  5795.4  433.08  5885.5  445.70  5915.4  448.29
#Mann=4,-1,0
  4158.1    0.05       0  4704.4    0.12       0  4986.1    0.03       0
  5004.6    0.05       0
Bank Sta=4616.2,5560.3
Exp/Cntr=0.3,0.1

Type RM Length L Ch R = 1,23911,1160,1160,1160
BEGIN DESCRIPTION:
ELM CREEK 20.0
END DESCRIPTION:
XS GIS Cut Line= 3
      2832725.02      7047175.00      2832025.00      7047275.00
      2830825.02      7047275.00
#Sta/Elev= 30
  4306.1  451.43  4578.9  446.34  4750.6  441.48  4770.8  440.25  4841.5  432.64
  4892.0  424.57  4950.5  418.33  4972.8  417.24  4982.9  414.55  4983.8  408.48
  4986.3  407.68  5002.3  408.48  5010.7  415.16  5015.7  415.16  5023.2  417.62
  5035.2  417.48  5143.2  415.19  5163.2  416.57  5313.2  414.94  5413.2  415.76
  5573.2  414.33  5623.2  415.37  5763.2  414.81  5812.4  418.33  5883.2  424.55
  6003.2  437.66  6073.2  441.72  6133.2  451.34  6153.2  452.58  6213.2  452.48
#Mann=4,-1,0
  4306.1    0.05       0  4983.8    0.07       0  5002.3    0.05       0
  5035.2    0.05       0
Bank Sta=4950.5,5812.4
Exp/Cntr=0.3,0.1

Type RM Length L Ch R = 1,22751,1029,1029,1029
BEGIN DESCRIPTION:
ELM CREEK 19.0
END DESCRIPTION:
XS GIS Cut Line= 3
      2832924.97      7046425.00      2831625.00      7046625.00
      2830824.97      7047225.02
#Sta/Elev= 30
  3636.1  461.03  3738.5  456.95  3865.0  448.78  4030.7  442.47  4212.8  432.09
  4264.6  429.93  4322.8  429.23  4391.1  426.07  4435.4  423.76  4465.7  420.84
  4475.8  420.62  4506.2  424.28  4527.7  424.83  4575.2  417.36  4597.2  415.02
  4668.1  413.88  4782.7  415.00  4959.4  415.84  4979.5  415.72  4992.1  409.65
  4994.6  408.85  5010.6  409.65  5014.9  414.51  5023.2  416.05  5258.7  412.11
  5414.9  414.80  5472.9  417.36  5758.7  437.60  5829.5  441.27  5951.4  451.26
#Mann=5,-1,0
  3636.1    0.05       0  4782.7    0.16       0  4959.4    0.05       0
  4992.1    0.03       0  5010.6    0.05       0
Bank Sta=4575.2,5472.9
Exp/Cntr=0.3,0.1

Type RM Length L Ch R = 1,21722,838,838,838
BEGIN DESCRIPTION:
ELM CREEK 18.0
END DESCRIPTION:
XS GIS Cut Line= 3
      2832425.03      7046175.00      2831225.00      7046175.00
      2830424.95      7046275.01
#Sta/Elev= 30
  3808.6  445.29  3978.6  436.72  4038.6  435.08  4158.6  428.17  4309.5  416.66
  4358.6  414.28  4388.6  413.78  4398.6  412.57  4418.6  413.42  4558.6  414.17
  4808.6  413.40  4968.6  414.60  4978.6  414.29  4988.6  410.17  4989.4  407.54
  4991.9  406.74  5005.4  406.74  5007.9  407.54  5008.6  408.35  5011.1  408.35
  5018.7  413.24  5026.5  413.86  5126.6  412.60  5149.7  412.71  5256.8  416.66
  5361.4  419.26  5421.8  421.71  5522.6  427.89  5734.2  442.80  5814.9  447.27
#Mann=5,-1,0
  3808.6    0.05       0  4989.4    0.03       0  5007.9    0.05       0
  5026.5    0.12       0  5126.6    0.05       0
Bank Sta=4309.5,5256.8
Exp/Cntr=0.3,0.1

Type RM Length L Ch R = 1,20884,1929,1929,1929
BEGIN DESCRIPTION:
ELM CREEK 17.0
END DESCRIPTION:
XS GIS Cut Line= 3
      2832774.97      7046124.99      2831075.00      7045425.00
      2830275.03      7046024.98
#Sta/Elev= 30
  3182.0  457.88  3327.2  453.40  3564.3  437.44  3772.1  435.27  3854.8  430.18
  3979.9  427.77  4068.8  423.70  4139.8  422.91  4236.9  416.38  4329.1  411.94
  4584.8  412.59  4620.3  412.17  4643.5  409.68  4674.4  412.52  4804.1  411.62
  4966.0  413.52  4981.8  413.69  5001.9  406.31  5004.4  405.51  5020.4  406.31
  5023.6  411.85  5027.7  413.78  5120.4  412.63  5261.3  414.42  5348.6  416.21
  5384.0  414.63  5428.2  416.38  5563.1  421.74  5856.9  442.82  6020.4  448.17
#Mann=5,-1,0
  3182.0    0.05       0  4966.0    0.12       0  5001.9    0.07       0
  5020.4    0.12       0  5261.3    0.05       0
Bank Sta=4236.9,5428.2
Exp/Cntr=0.3,0.1

Type RM Length L Ch R = 1,18955,1523,1523,1523
BEGIN DESCRIPTION:
ELM CREEK 16.0
END DESCRIPTION:
XS GIS Cut Line= 3
      2831025.00      7043674.98      2831025.00      7044375.00
      2830224.98      7045825.03
#Sta/Elev= 30
  4307.7  449.83  4432.3  449.26  4497.7  445.10  4707.7  424.47  4820.1  415.60
  4887.7  411.60  4977.7  410.89  4987.7  408.94  4995.9  403.97  4998.4  403.17
  5014.5  403.97  5015.7  409.92  5021.5  410.99  5102.8  411.04  5124.6  408.15
  5140.7  410.60  5200.3  411.38  5265.6  410.26  5361.8  411.55  5368.7  410.16
  5384.6  411.65  5612.9  411.41  5624.5  412.80  5662.1  411.18  6090.0  411.87
  6178.6  415.60  6297.0  421.55  6465.5  433.82  6568.6  439.72  6663.8  442.67
#Mann=5,-1,0
  4307.7    0.16       0  4432.3    0.12       0  4995.9    0.07       0
  5014.5    0.12       0  6090.0    0.05       0
Bank Sta=4820.1,6178.6
Exp/Cntr=0.3,0.1

Type RM Length L Ch R = 1,17432,1119,1119,1119
BEGIN DESCRIPTION:
double ELM CREEK 15.0
END DESCRIPTION:
XS GIS Cut Line= 3
      2830819.31      7043693.13      2830003.35      7044179.23
      2829275.00      7044475.00
#Sta/Elev= 30
  4239.6  445.96  4411.4  436.46  4543.8  434.75  4682.0  436.56  4746.2  431.51
  4820.2  428.18  4835.8  429.34  4841.6  427.55  4854.5  427.35  4931.2  422.43
  4958.5  418.75  4969.2  414.82  4979.9  407.92  4980.3  403.18  4982.8  402.38
  4998.9  403.18  5001.3  405.45  5011.0  406.53  5016.9  409.96  5024.5  410.72
  5139.5  409.56  5489.8  410.63  5554.6  412.43  5591.2  408.54  5597.7  411.17
  5608.5  412.26  5630.1  411.57  5677.2  414.82  5853.6  436.51  5975.5  446.48
#Mann=5,-1,0
  4239.6    0.16       0  4854.5    0.12       0  4980.3    0.07       0
  4998.9    0.12       0  5139.5    0.05       0
Bank Sta=4969.2,5677.2
Exp/Cntr=0.3,0.1

Type RM Length L Ch R = 1,16313,1852,1852,1852
BEGIN DESCRIPTION:
double ELM CREEK 14.0
END DESCRIPTION:
XS GIS Cut Line= 3
      2830925.03      7043625.00      2830289.81      7043554.23
      2829025.00      7043125.00
#Sta/Elev= 30
  4364.2  449.02  4494.8  445.12  4595.6  437.10  4675.7  434.05  4817.0  422.38
  4940.0  415.86  4968.3  414.13  4988.1  407.91  4994.0  402.26  4996.5  401.46
  5012.6  402.26  5029.5  409.40  5092.9  407.44  5140.7  409.88  5203.5  409.39
  5219.6  405.19  5234.9  405.53  5240.7  408.26  5251.3  409.30  5378.0  408.22
  5391.9  403.31  5399.2  407.41  5409.7  409.00  5467.7  409.62  5729.4  414.13
  5991.7  421.87  6066.3  425.07  6108.8  427.33  6234.4  440.87  6339.0  447.46
#Mann=7,-1,0
  4364.2    0.16       0  4940.0    0.12       0  4994.0    0.07       0
  5012.6    0.12       0  5467.7    0.05       0  5991.7    0.16       0
  6066.3    0.05       0
Bank Sta=4968.3,5729.4
Exp/Cntr=0.3,0.1

Type RM Length L Ch R = 1,14461,617,617,617
BEGIN DESCRIPTION:
ELM CREEK 13.0
END DESCRIPTION:
XS GIS Cut Line= 3
      2831074.96      7043274.98      2830271.68      7042837.49
      2829574.98      7042875.00
#Sta/Elev= 30
  3959.6  447.65  4033.2  442.60  4187.3  425.50  4289.3  417.16  4368.8  411.99
  4469.0  408.14  4654.2  408.96  4676.1  408.12  4681.7  404.79  4697.9  407.12
  4703.6  403.19  4711.1  402.98  4747.3  402.92  4763.4  407.90  4845.1  407.99
  4871.7  405.08  4911.0  407.58  4981.1  407.69  4991.1  403.76  4991.6  400.59
  4994.1  399.79  5010.8  400.59  5031.2  406.84  5118.6  411.82  5120.7  411.99
  5289.8  433.02  5361.7  439.68  5421.8  442.36  5549.4  443.71  5572.0  443.63
#Mann=6,-1,0
  3959.6    0.16       0  4289.3    0.12       0  4991.6    0.07       0
  5010.8    0.12       0  5118.6    0.16       0  5549.4    0.05       0
Bank Sta=4368.8,5120.7
Exp/Cntr=0.3,0.1

Type RM Length L Ch R = 1,13844,343,343,343
BEGIN DESCRIPTION:
ELM CREEK 12.0
END DESCRIPTION:
XS GIS Cut Line= 3
      2831074.99      7043174.99      2830375.00      7042375.00
      2829675.00      7042375.00
#Sta/Elev= 30
  3934.5  444.64  4140.0  422.95  4237.8  414.73  4283.4  410.90  4366.8  406.72
  4501.6  407.72  4544.3  406.09  4565.2  407.68  4579.4  406.61  4678.6  406.19
  4820.5  407.38  4849.0  406.17  4855.6  407.07  4961.9  407.69  4969.5  406.90
  4976.1  401.71  4980.8  400.66  4983.3  399.86  5000.0  400.66  5007.5  401.03
  5027.5  406.59  5037.5  407.72  5077.5  407.61  5166.4  410.90  5177.5  412.50
  5217.5  414.44  5363.8  419.52  5462.8  426.26  5597.5  436.48  5697.5  440.05
#Mann=6,-1,0
  3934.5    0.16       0  4237.8    0.12       0  4980.8    0.07       0
  5000.0    0.12       0  5363.8    0.16       0  5462.8    0.05       0
Bank Sta=4283.4,5166.4
Exp/Cntr=0.3,0.1

Type RM Length L Ch R = 1,13501,819,819,819
BEGIN DESCRIPTION:
Mapping XS f5c01a00
END DESCRIPTION:
XS GIS Cut Line= 3
      2831738.33      7043248.61      2830592.47      7042097.55
      2829718.78      7042081.94
#Sta/Elev= 30
  3305.3  446.74  3331.4  447.15  3352.6  445.39  3536.5  440.91  3614.3  435.55
  3706.2  432.52  3832.4  421.16  3918.3  414.55  4047.4  410.37  4208.2  406.99
  4314.3  407.61  4554.7  406.30  4568.8  405.19  4759.8  405.28  4956.9  407.52
  4977.4  400.40  4979.9  399.60  4996.6  400.40  5017.0  402.24  5027.0  407.14
  5047.0  410.26  5167.0  408.66  5304.1  410.37  5308.5  410.53  5397.0  412.06
  5550.5  417.94  5657.1  421.71  5734.0  427.74  5743.8  428.66  5803.3  433.84
#Mann=8,-1,0
  3305.3    0.16       0  3832.4    0.12       0  4977.4    0.07       0
  4996.6    0.12       0  5308.5    0.05       0  5550.5    0.16       0
  5734.0    0.12       0  5743.8    0.16       0
Bank Sta=4047.4,5304.1
Exp/Cntr=0.3,0.1

Type RM Length L Ch R = 1,12682,955,955,955
BEGIN DESCRIPTION:
double ELM CREEK 11.0
END DESCRIPTION:
XS GIS Cut Line= 3
      2831686.21      7040482.98      2830575.00      7041775.00
      2829674.98      7041875.00
#Sta/Elev= 30
  3284.0  445.23  3399.8  439.76  3516.2  444.28  3619.3  447.34  3750.3  445.23
  3867.3  435.17  4073.6  412.87  4094.4  413.56  4143.4  409.66  4256.2  406.47
  4297.1  405.13  4364.3  404.65  4370.9  403.17  4382.7  404.50  4548.2  404.07
  4938.2  407.12  4974.4  406.78  4988.6  400.45  4991.1  399.65  5007.8  400.45
  5018.3  406.57  5209.5  406.01  5338.0  409.66  5379.6  410.36  5541.5  412.04
  5662.3  418.10  5745.0  424.62  5844.9  433.91  5874.9  436.29  5893.7  437.16
#Mann=13,-1,0
  3284.0    0.16       0  3516.2    0.05       0  3750.3    0.16       0
  4256.2    0.12       0  4297.1    0.07       0  4382.7    0.05       0
  4548.2    0.12       0  4988.6    0.07       0  5007.8    0.12       0
  5379.6    0.05       0  5745.0    0.12       0  5844.9    0.16       0
  5874.9    0.12       0
Bank Sta=4143.4,5338
Exp/Cntr=0.3,0.1

Type RM Length L Ch R = 1,11727,897,897,897
BEGIN DESCRIPTION:
double ELM CREEK 10.0
END DESCRIPTION:
XS GIS Cut Line= 3
      2831175.01      7040725.00      2830175.00      7041225.00
      2829375.04      7041524.99
#Sta/Elev= 30
  3834.0  444.89  3877.0  441.94  4035.3  427.38  4183.4  416.63  4337.0  408.87
  4357.1  407.49  4490.9  404.02  4518.8  400.91  4557.9  404.33  4653.0  403.23
  4826.3  405.49  4854.2  405.36  4862.6  401.14  4871.0  400.72  4928.5  400.53
  4931.0  399.73  4947.7  400.53  4949.2  403.27  4961.8  402.13  4967.2  405.20
  4984.1  401.31  5005.4  400.98  5016.1  405.82  5022.4  406.08  5027.7  403.47
  5263.5  408.87  5291.6  410.85  5407.9  417.89  5742.5  437.64  5806.4  440.38
#Mann=8,-1,0
  3834.0    0.05       0  3877.0    0.16       0  4357.1    0.12       0
  4928.5    0.07       0  4947.7    0.12       0  5291.6    0.05       0
  5407.9    0.16       0  5742.5    0.05       0
Bank Sta=4337,5263.5
Exp/Cntr=0.3,0.1

Type RM Length L Ch R = 1,10830,672,672,672
BEGIN DESCRIPTION:
Mapping XS df4c70d7
END DESCRIPTION:
XS GIS Cut Line= 3
      2831131.86      7040385.81      2830272.45      7040715.69
      2829473.86      7041114.98
#Sta/Elev= 30
  4098.3  436.14  4112.2  436.77  4195.2  440.34  4225.2  439.55  4304.6  431.17
  4309.9  431.79  4364.6  427.06  4480.5  421.25  4496.2  417.72  4512.7  416.74
  4523.3  419.10  4558.7  417.57  4588.7  414.54  4608.0  414.82  4787.7  408.07
  4906.2  405.12  4941.1  404.47  4952.2  402.69  4971.5  402.90  4974.3  400.27
  4976.8  399.47  4993.7  400.27  5006.9  400.55  5014.8  403.24  5030.6  404.75
  5190.1  404.05  5552.6  403.32  5653.1  408.07  5785.3  413.85  5911.7  423.45
#Mann=7,-1,0
  4098.3    0.05       0  4112.2    0.08       0  4496.2    0.16       0
  4906.2    0.12       0  4974.3    0.07       0  4993.7    0.12       0
  5190.1    0.05       0
Bank Sta=4787.7,5653.1
Exp/Cntr=0.3,0.1

Type RM Length L Ch R = 1,10158,190,190,190
BEGIN DESCRIPTION:
Mapping XS 80e4fdba
END DESCRIPTION:
XS GIS Cut Line= 3
      2830836.65      7040194.86      2829890.50      7040272.98
      2828822.75      7040316.38
#Sta/Elev= 30
  4075.6  432.49  4207.7  430.12  4377.2  430.25  4478.6  423.36  4558.9  416.37
  4609.1  413.70  4649.2  409.46  4687.2  407.60  4709.4  405.83  4789.7  403.27
  4809.7  400.72  4829.8  400.76  4849.9  403.50  4960.2  403.78  4970.6  400.26
  4973.1  399.46  4990.1  400.26  5025.0  400.26  5032.2  401.21  5040.5  402.80
  5080.5  403.56  5201.7  402.33  5444.9  403.82  5518.4  407.60  5693.1  411.70
  5781.1  412.36  5886.2  416.32  5994.1  420.38  6061.3  422.54  6093.6  424.68
#Mann=6,-1,0
  4075.6    0.08       0  4970.6    0.04       0  4990.1    0.08       0
  5032.2    0.08       0  5886.2    0.05       0  5994.1    0.08       0
Bank Sta=4687.2,5518.4
Exp/Cntr=0.3,0.1

Type RM Length L Ch R = 1,9968,724,724,724
BEGIN DESCRIPTION:
Mapping XS fdca467a
END DESCRIPTION:
XS GIS Cut Line= 3
      2830628.34      7040047.28      2829899.18      7040082.01
      2828798.38      7040108.01
#Sta/Elev= 30
  4272.8  438.29  4274.5  438.29  4286.9  438.10  4346.2  435.85  4476.4  427.34
  4486.4  426.29  4506.4  419.49  4535.8  416.09  4540.8  417.18  4606.5  413.00
  4729.6  409.10  4799.6  407.27  4856.8  405.34  4938.4  404.53  4956.3  405.04
  4977.2  400.26  4979.7  399.46  4996.7  400.26  5027.0  400.94  5037.6  403.62
  5446.6  405.39  5527.1  406.58  5647.2  405.45  5731.5  407.01  5741.5  407.27
  5918.8  412.75  5967.2  415.65  5977.2  417.28  6027.3  416.59  6103.9  420.35
#Mann=11,-1,0
  4272.8    0.08       0  4274.5     0.1       0  4286.9    0.08       0
  4729.6    0.05       0  4938.4     0.1       0  4977.2    0.07       0
  4996.7     0.1       0  5037.6    0.12       0  5446.6    0.05       0
  5731.5    0.08       0  5918.8    0.05       0
Bank Sta=4799.6,5741.5
Exp/Cntr=0.3,0.1

Type RM Length L Ch R = 1,9244,1239,1239,1239
BEGIN DESCRIPTION:
Mapping XS eb80dca0
END DESCRIPTION:
XS GIS Cut Line= 3
      2830862.70      7038970.91      2829673.49      7039430.96
      2828798.74      7039959.28
#Sta/Elev= 30
  3704.5  427.30  3820.0  421.01  4080.4  411.12  4206.1  406.35  4225.3  407.38
  4248.9  406.03  4260.6  407.09  4430.0  405.13  4448.8  403.79  4709.9  401.28
  4806.1  401.88  4917.6  402.03  4974.8  403.66  4979.8  400.26  4982.3  399.46
  4999.3  400.26  5011.7  400.28  5017.6  402.65  5024.6  403.26  5176.7  402.79
  5192.2  401.82  5330.0  402.15  5410.1  404.19  5439.5  403.58  5518.0  401.44
  5556.9  401.55  5641.0  405.13  5674.3  406.46  5867.2  414.16  6001.5  417.55
#Mann=11,-1,0
  3704.5    0.16       0  4080.4    0.12       0  4806.1    0.05       0
  4917.6    0.12       0  4979.8    0.07       0  4999.3    0.12       0
  5439.5     0.1       0  5518.0    0.08       0  5556.9    0.05       0
  5674.3    0.08       0  5867.2    0.05       0
Bank Sta=4430,5641
Exp/Cntr=0.3,0.1

Type RM Length L Ch R = 1,8005,636,636,636
BEGIN DESCRIPTION:
Mapping XS 8df110ae
END DESCRIPTION:
XS GIS Cut Line= 3
      2829187.38      7038007.36      2828970.37      7038727.84
      2828683.91      7039838.95
#Sta/Elev= 30
  4268.7  421.91  4293.3  421.61  4298.5  422.85  4359.3  423.23  4364.5  424.05
  4397.5  422.84  4435.8  424.66  4468.8  425.11  4516.9  423.72  4573.0  419.83
  4631.8  414.39  4707.5  403.80  4714.2  402.80  4748.5  400.88  4757.7  399.21
  4760.2  398.41  4774.8  398.41  4777.3  399.21  4815.6  399.21  4892.0  399.21
  5119.0  399.21  5338.1  399.21  5348.7  400.78  5490.7  401.22  5609.4  403.80
  5699.1  407.55  5943.2  414.37  5983.9  413.75  6024.6  414.44  6168.6  420.88
#Mann=8,-1,0
  4268.7    0.05       0  4714.2    0.16       0  4757.7   0.033       0
  4777.3    0.16       0  4815.6    0.07       0  4892.0    0.05       0
  5119.0    0.07       0  5490.7    0.05       0
Bank Sta=4707.5,5609.4
Exp/Cntr=0.3,0.1

Type RM Length L Ch R = 1,7369,901,901,901
BEGIN DESCRIPTION:
Mapping XS 1921f685
END DESCRIPTION:
XS GIS Cut Line= 3
      2828640.52      7037868.44      2828423.49      7038389.30
      2828510.27      7039630.30
#Sta/Elev= 30
  4431.7  434.21  4480.9  431.46  4510.1  428.37  4534.0  427.04  4539.4  425.11
  4557.8  424.65  4579.6  422.63  4610.9  419.41  4640.1  414.59  4655.5  413.63
  4669.4  410.50  4687.8  409.17  4698.8  407.05  4712.9  405.79  4728.1  403.50
  4740.9  401.09  4743.2  399.21  4745.7  398.41  4760.3  398.41  4762.8  399.21
  5351.0  399.21  5432.7  399.21  5442.8  400.39  5556.7  401.59  5653.3  402.03
  5743.1  403.50  5783.6  404.64  5843.7  408.21  6014.1  411.41  6240.0  419.74
#Mann=6,-1,0
  4431.7    0.16       0  4712.9    0.05       0  4743.2   0.033       0
  4762.8    0.05       0  5351.0    0.07       0  5556.7    0.05       0
Bank Sta=4728.1,5743.1
Exp/Cntr=0.3,0.1

Type RM Length L Ch R = 1,6468,818,818,818
BEGIN DESCRIPTION:
ELM CREEK 4.0
END DESCRIPTION:
XS GIS Cut Line= 3
      2828475.00      7037475.00      2827575.00      7038075.00
      2827575.00      7039275.03
#Sta/Elev= 30
  3929.3  441.74  3987.9  440.88  4023.9  438.00  4138.1  426.08  4153.1  423.64
  4195.2  419.76  4240.3  412.42  4246.3  412.41  4267.3  407.70  4317.5  403.24
  4335.1  401.40  4354.5  400.66  4359.6  399.21  4362.1  398.41  4376.9  398.41
  4379.4  399.21  4382.6  399.21  4456.0  399.21  5471.0  399.21  5486.9  403.24
  5491.0  404.68  5681.0  415.70  5731.0  419.80  5791.0  419.93  5801.0  420.28
  5811.0  422.66  5821.0  423.51  5911.0  425.47  6081.0  431.54  6211.0  435.00
#Mann=6,-1,0
  3929.3    0.16       0  4335.1    0.05       0  4359.6   0.033       0
  4379.4    0.05       0  4382.6    0.07       0  4456.0    0.05       0
Bank Sta=4317.5,5486.9
Exp/Cntr=0.3,0.1

Type RM Length L Ch R = 1,5650,806,806,806
BEGIN DESCRIPTION:
ELM CREEK 3.0
END DESCRIPTION:
XS GIS Cut Line= 3
      2826925.00      7036774.96      2826825.00      7037775.00
      2826525.00      7039174.99
#Sta/Elev= 30
  4007.2  440.53  4055.0  441.88  4097.7  437.92  4208.2  420.34  4340.7  403.08
  4356.5  400.52  4359.1  399.21  4361.6  398.41  4376.4  398.41  4378.9  399.21
  5728.1  399.21  5738.3  399.44  5747.7  400.82  5769.0  400.90  5817.4  403.08
  5846.6  404.65  6014.5  407.85  6083.5  410.04  6127.0  407.96  6138.1  411.75
  6208.8  415.42  6231.8  417.42  6249.7  420.37  6270.2  420.59  6311.1  425.04
  6352.0  427.59  6369.9  430.20  6382.7  430.59  6413.3  433.78  6444.0  435.28
#Mann=3,-1,0
  4007.2    0.05       0  4359.1   0.033       0  4378.9    0.05       0
Bank Sta=4340.7,5817.4
Exp/Cntr=0.3,0.1

Type RM Length L Ch R = 1,4844,981,981,981
BEGIN DESCRIPTION:
ELM CREEK 2.0
END DESCRIPTION:
XS GIS Cut Line= 3
      2826825.04      7036774.97      2826125.00      7037375.00
      2824925.00      7037875.00
#Sta/Elev= 30
  4070.4  440.01  4112.7  437.08  4176.4  428.93  4212.6  425.52  4247.7  420.70
  4290.5  416.59  4339.9  410.53  4382.7  407.61  4389.3  406.18  4425.5  403.80
  4428.8  402.95  4432.1  402.10  4446.4  401.60  4457.3  399.21  4459.8  398.41
  4474.6  398.41  4477.1  399.21  5946.3  399.21  5981.6  402.95  6047.0  410.00
  6070.9  414.33  6094.7  416.77  6100.1  416.57  6118.5  419.71  6123.9  419.42
  6147.8  423.41  6153.2  423.50  6177.0  426.64  6224.7  433.67  6292.4  437.07
#Mann=3,-1,0
  4070.4    0.05       0  4457.3   0.033       0  4477.1    0.05       0
Bank Sta=4428.8,5981.6
Exp/Cntr=0.3,0.1

Type RM Length L Ch R = 1,3863,967,967,967
BEGIN DESCRIPTION:
Mapping XS f7919cc6
END DESCRIPTION:
XS GIS Cut Line= 3
      2826867.66      7036110.49      2825526.56      7036553.18
      2824667.96      7037710.98
#Sta/Elev= 30
  3403.6  439.23  3427.5  439.56  3543.3  433.39  3592.1  427.58  3617.0  426.34
  3859.2  426.36  3869.8  427.09  3883.1  431.58  3901.3  431.49  3909.5  430.15
  3914.8  424.63  4004.8  425.72  4010.1  424.43  4036.5  425.05  4041.8  423.56
  4131.8  422.52  4352.7  402.74  4375.9  399.21  4378.4  398.41  4395.7  399.21
  5613.0  399.21  5682.3  402.74  5683.8  402.96  5804.2  411.80  5833.5  412.32
  5868.9  415.81  5904.4  421.74  6025.8  428.92  6184.1  435.30  6257.3  434.60
#Mann=5,-1,0
  3403.6    0.05       0  4375.9   0.033       0  4395.7    0.05       0
  5613.0    0.07       0  5683.8    0.05       0
Bank Sta=4352.7,5682.3
Exp/Cntr=0.3,0.1

Type RM Length L Ch R = 1,2896,734,734,734
BEGIN DESCRIPTION:
Mapping XS 9b4487f2
END DESCRIPTION:
XS GIS Cut Line= 3
      2827440.66      7035719.84      2824992.70      7035797.97
      2823378.11      7037152.14
#Sta/Elev= 30
  2375.0  438.74  2840.9  437.72  2997.3  438.90  3261.1  438.27  3341.2  439.92
  3941.5  438.08  4121.6  425.57  4231.6  419.77  4407.8  406.12  4443.3  402.90
  4447.7  402.39  4471.8  399.21  4474.3  398.41  4491.7  399.21  5579.5  399.21
  5633.1  402.39  5643.5  405.38  5757.7  412.68  5778.6  410.65  5786.3  414.41
  5850.1  419.15  6098.6  430.96  6197.5  430.22  6289.8  433.11  6310.7  430.51
  6382.2  435.23  6744.1  437.81  6776.1  438.73  6892.4  437.19  6931.5  437.04
#Mann=9,-1,0
  2375.0    0.16       0  2997.3    0.05       0  4407.8    0.16       0
  4443.3    0.05       0  4471.8   0.033       0  4491.7    0.05       0
  6744.1    0.16       0  6776.1    0.12       0  6892.4    0.05       0
Bank Sta=4447.7,5633.1
Exp/Cntr=0.3,0.1

Type RM Length L Ch R = 1,2162,1844,1844,1844
BEGIN DESCRIPTION:
Mapping XS 5d95762f
END DESCRIPTION:
XS GIS Cut Line= 3
      2827063.07      7035563.60      2824315.62      7035316.20
      2823339.54      7036864.91
#Sta/Elev= 30
  2342.0  438.17  2611.1  438.92  2721.6  433.48  2751.7  429.23  2771.8  432.99
  2882.2  439.40  3263.8  437.87  3434.5  426.81  3454.5  421.64  3474.6  426.17
  3493.4  427.23  3609.4  431.80  3675.4  437.07  3745.7  438.03  3926.4  433.15
  4093.4  418.45  4192.7  408.15  4244.2  402.03  4257.8  401.60  4265.3  399.21
  4267.8  398.41  4285.2  399.21  5651.9  399.21  5706.5  402.03  5876.7  410.67
  5913.2  415.57  5992.1  421.28  6311.1  435.52  6703.0  436.30  6931.2  433.77
#Mann=5,-1,0
  2342.0    0.16       0  4093.4    0.12       0  4192.7    0.05       0
  4265.3   0.033       0  4285.2    0.05       0
Bank Sta=4244.2,5706.5
Exp/Cntr=0.3,0.1

Type RM Length L Ch R = 1,318,0,0,0
BEGIN DESCRIPTION:
ELM CREEK 1.0
END DESCRIPTION:
XS GIS Cut Line= 3
      2826516.19      7033962.03      2823284.61      7033869.83
      2823070.87      7037207.99
#Sta/Elev= 30
  1767.1  438.10  1858.3  436.94  1950.2  430.55  1988.4  429.53  2041.8  425.21
  2228.5  413.55  2378.5  412.43  2428.6  410.71  2498.6  404.93  2534.3  400.37
  2536.9  399.94  2538.6  399.21  2541.1  398.41  2558.6  399.21  6572.3  399.94
  6738.7  401.29  6787.6  404.00  6899.1  406.92  7134.3  419.02  7186.8  421.34
  7263.9  423.13  7309.9  425.70  7450.2  424.61  7560.4  420.48  7720.7  421.25
  7740.8  419.51  7810.9  419.01  7864.4  420.79  8046.0  423.02  8345.0  431.61
#Mann=10,-1,0
  1767.1    0.16       0  1950.2    0.05       0  2041.8    0.16       0
  2534.3    0.05       0  2538.6   0.033       0  2558.6    0.05       0
  6787.6     0.1       0  7134.3    0.05       0  7186.8    0.16       0
  7864.4    0.05       0
Bank Sta=2536.9,6572.3
Exp/Cntr=0.3,0.1

Chan Stop Cuts=-1
