--- Penson Spring Branch.prj (project) ---

Proj Title=Penson Spring Branch Base Level Engineering
Current Plan=p01
Default Exp/Contr=0.3,0.1
English Units
Geom File=g01
Flow File=f01
Plan File=p01
BEGIN DESCRIPTION:
Penson Spring Branch
END DESCRIPTION:

--- Penson Spring Branch.p01 (plan) ---

Plan Title=Multiple Run
Short Identifier=Multiple
Geom File=g01
Flow File=f01
Subcritical Flow
K Sum by GR= 0
Std Step Tol= 0.01
Critical Tol= 0.01
Num of Std Step Trials= 20
Max Error Tol= 0.3
Flow Tol Ratio= 0.001
Split Flow NTrial= 30
Split Flow Tol= 0.02
Split Flow Ratio= 0.02
Log Output Level= 0
Friction Slope Method= 1
Unsteady Friction Slope Method= 2
Unsteady Bridges Friction Slope Method= 1
Parabolic Critical Depth
Global Vel Dist=  1 , 1 , 1
Global Log Level= 0
CheckData=True
Encroach Param= -1, 0, 0, 0
BEGIN DESCRIPTION:
Multiple Run
END DESCRIPTION:

--- Penson Spring Branch.f01 (steady flow) ---

Flow Title=Multiple
Number of Profiles=7
Profile Names=10-year,25-year,50-year,1pct_min,100-year,1pct_plu,500-year
River Rch & RM= Penson Spring Br,Reach-1,23318
     348     449     529     310     618    1234     846
River Rch & RM= Penson Spring Br,Reach-1,16361
     608     811     975     582    1162    2319    1653
River Rch & RM= Penson Spring Br,Reach-1,10302
     806    1087    1316     790    1577    3147    2269
River Rch & RM= Penson Spring Br,Reach-1,4753
     949    1283    1556     936    1867    3724    2691
Boundary for River Rch & Prof#=Penson Spring Br,Reach-1,1
Up Type=0
Dn Type=3
Dn Slope=0.005
Boundary for River Rch & Prof#=Penson Spring Br,Reach-1,2
Up Type=0
Dn Type=3
Dn Slope=0.005
Boundary for River Rch & Prof#=Penson Spring Br,Reach-1,3
Up Type=0
Dn Type=3
Dn Slope=0.005
Boundary for River Rch & Prof#=Penson Spring Br,Reach-1,4
Up Type=0
Dn Type=3
Dn Slope=0.005
Boundary for River Rch & Prof#=Penson Spring Br,Reach-1,5
Up Type=0
Dn Type=3
Dn Slope=0.005
Boundary for River Rch & Prof#=Penson Spring Br,Reach-1,6
Up Type=0
Dn Type=3
Dn Slope=0.005
Boundary for River Rch & Prof#=Penson Spring Br,Reach-1,7
Up Type=0
Dn Type=3
Dn Slope=0.005

--- Penson Spring Branch.g01 (geometry) ---

Geom Title=Existing Conditions

River Reach=Penson Spring Br,Reach-1
Reach XY= 30
      2827316.67      7012423.35      2827884.81      7012480.90
      2828442.40      7012879.47      2828578.51      7013470.44
      2828819.49      7013764.19      2829320.67      7013611.76
      2829870.91      7013801.20      2830402.92      7013579.62
      2830688.90      7013634.30      2831224.56      7014061.69
      2831440.10      7014476.00      2832056.71      7014756.18
      2832215.05      7014599.87      2832682.75      7015505.98
      2833073.62      7015687.46      2833425.05      7015499.41
      2833965.69      7015950.91      2834757.47      7016245.46
      2834874.85      7016584.48      2835044.70      7016472.62
      2835278.08      7016646.62      2835631.59      7016380.79
      2835924.35      7016934.54      2836596.86      7017140.30
      2837073.28      7017098.88      2837383.67      7017345.46
      2839422.51      7016756.89      2840329.75      7016929.24
      2841695.48      7017413.75      2844859.00      7019148.24

Type RM Length L Ch R = 1,23318,245,245,245
BEGIN DESCRIPTION:
Mapping XS a031f925
END DESCRIPTION:
XS GIS Cut Line= 3
      2827423.96      7012836.62      2827450.72      7012408.35
      2827257.41      7011974.14
#Sta/Elev= 30
  4586.7  473.61  4618.4  473.07  4628.4  473.27  4668.5  472.12  4758.7  470.63
  4908.9  469.13  4954.8  468.93  4980.0  468.78  4989.1  467.89  4996.1  466.74
  4996.6  465.94  5001.6  465.94  5002.1  466.74  5004.2  467.68  5009.2  467.74
  5015.0  468.45  5030.4  468.66  5044.5  468.54  5062.3  467.37  5068.7  467.43
  5074.2  468.00  5085.1  468.45  5096.5  468.38  5107.0  467.70  5114.2  467.66
  5194.9  468.12  5259.1  468.09  5316.6  468.51  5427.7  468.78  5491.1  469.66
#Mann=5,-1,0
  4586.7    0.05       0  4954.8    0.08       0  4996.1    0.07       0
  5002.1    0.08       0  5068.7    0.05       0
Bank Sta=4980,5427.7
Exp/Cntr=0.3,0.1

Type RM Length L Ch R = 1,23073,320,320,320
BEGIN DESCRIPTION:
Mapping XS 96172f62
END DESCRIPTION:
XS GIS Cut Line= 3
      2827554.56      7013007.18      2827702.37      7012403.67
      2827527.03      7012038.53
#Sta/Elev= 30
  4413.5  473.56  4475.4  473.05  4480.5  472.75  4522.1  472.05  4558.6  471.90
  4745.2  469.03  4837.9  468.10  4927.2  467.63  4951.1  468.37  4979.8  466.89
  4992.3  466.84  4999.6  466.19  5000.1  465.39  5005.1  465.39  5005.6  466.19
  5012.9  467.62  5021.4  468.57  5031.6  468.83  5045.2  468.70  5055.6  467.90
  5062.3  466.60  5067.8  466.56  5077.7  467.16  5099.9  467.08  5107.5  466.84
  5130.2  467.09  5266.1  466.99  5322.4  467.31  5339.5  467.17  5439.9  467.45
#Mann=3,-1,0
  4413.5    0.05       0  4999.6    0.04       0  5005.6    0.05       0
Bank Sta=4927.2,5439.9
Exp/Cntr=0.3,0.1

Type RM Length L Ch R = 1,22753,391,391,391
BEGIN DESCRIPTION:
Mapping XS 5185f28b
END DESCRIPTION:
XS GIS Cut Line= 3
      2827850.44      7013037.70      2827981.37      7012563.98
      2828184.19      7012139.86
#Sta/Elev= 30
  4475.2  468.58  4547.0  468.74  4626.1  467.84  4694.7  467.66  4699.9  468.02
  4707.1  467.49  4768.5  466.60  4782.4  465.93  4887.1  464.75  4913.7  465.00
  4934.5  465.94  4990.0  464.59  4998.8  463.80  5029.3  464.48  5040.1  463.64
  5040.6  462.84  5045.6  462.84  5046.1  463.64  5052.5  464.31  5080.7  464.49
  5103.3  466.01  5109.6  467.84  5120.5  468.45  5142.9  468.19  5148.7  466.85
  5153.9  466.70  5165.1  465.79  5260.3  465.93  5352.8  467.11  5436.8  469.79
#Mann=6,-1,0
  4475.2    0.05       0  4707.1    0.16       0  5029.3    0.08       0
  5040.1    0.07       0  5046.1    0.08       0  5153.9    0.05       0
Bank Sta=4782.4,5260.3
Exp/Cntr=0.3,0.1

Type RM Length L Ch R = 1,22362,354,354,354
BEGIN DESCRIPTION:
Mapping XS c18e8fc7
END DESCRIPTION:
XS GIS Cut Line= 3
      2827939.39      7013178.79      2828282.30      7012818.52
      2828356.09      7012430.04
#Sta/Elev= 30
  4463.1  467.42  4575.9  466.84  4766.9  465.03  4848.4  463.95  4876.5  463.66
  4929.5  463.75  4943.6  463.55  4960.5  462.64  5000.7  461.94  5005.8  462.18
  5053.0  462.16  5055.0  461.77  5055.5  460.97  5060.5  460.97  5061.0  461.77
  5096.4  461.93  5105.2  462.40  5126.9  462.78  5137.1  462.36  5157.4  462.35
  5204.6  463.95  5220.7  464.59  5249.1  465.86  5267.0  465.91  5272.1  466.40
  5279.6  466.23  5300.0  466.57  5324.3  466.04  5340.7  468.18  5355.9  468.64
#Mann=5,-1,0
  4463.1    0.05       0  4876.5    0.16       0  5055.0    0.07       0
  5061.0    0.16       0  5220.7    0.08       0
Bank Sta=4848.4,5204.6
Exp/Cntr=0.3,0.1

Type RM Length L Ch R = 1,22008,391,391,391
BEGIN DESCRIPTION:
Mapping XS 156e23c9
END DESCRIPTION:
XS GIS Cut Line= 3
      2827965.44      7013289.45      2828514.50      7013055.07
      2828842.21      7012497.31
#Sta/Elev= 30
  4365.6  466.95  4690.6  463.45  4725.1  463.64  4748.2  462.89  4764.9  461.98
  4778.3  461.07  4810.9  460.74  4843.1  462.30  4908.8  461.62  4930.5  462.30
  4971.0  461.03  4992.4  459.45  4995.2  458.54  4995.7  457.74  5000.7  457.74
  5001.2  458.54  5013.9  460.00  5044.4  460.67  5078.7  461.32  5094.0  462.32
  5153.5  461.98  5156.4  462.05  5172.2  462.38  5328.4  464.19  5410.3  466.53
  5461.3  468.21  5476.2  468.10  5530.1  469.88  5590.1  472.58  5609.5  472.14
#Mann=10,-1,0
  4365.6    0.05       0  4748.2    0.16       0  4995.2    0.07       0
  5001.2    0.16       0  5044.4    0.05       0  5156.4    0.08       0
  5172.2    0.05       0  5410.3    0.08       0  5476.2    0.05       0
  5530.1    0.08       0
Bank Sta=4764.9,5153.5
Exp/Cntr=0.3,0.1

Type RM Length L Ch R = 1,21617,305,305,305
BEGIN DESCRIPTION:
Mapping XS 64b09535
END DESCRIPTION:
XS GIS Cut Line= 4
      2828100.40      7013528.60      2828579.61      7013365.40
      2828857.38      7013236.92      2828996.29      7012941.75
#Sta/Elev= 30
  4529.4  465.30  4671.6  463.81  4762.2  463.69  4872.3  461.80  4937.3  459.07
  4974.9  456.01  4975.4  455.21  4980.4  455.21  4980.9  456.01  4992.1  456.77
  5023.4  456.88  5062.4  459.07  5089.6  460.18  5173.8  461.92  5213.8  463.53
  5295.0  464.97  5365.8  464.64  5377.0  463.99  5394.2  464.10  5421.7  463.36
  5445.3  462.52  5462.6  462.50  5472.5  461.87  5485.3  461.01  5520.6  460.48
  5575.9  461.14  5582.1  462.68  5604.8  461.98  5633.2  462.06  5667.9  463.35
#Mann=7,-1,0
  4529.4    0.05       0  4762.2    0.16       0  4974.9    0.07       0
  4980.9    0.16       0  5089.6    0.05       0  5421.7    0.08       0
  5472.5    0.05       0
Bank Sta=4937.3,5062.4
Exp/Cntr=0.3,0.1

Type RM Length L Ch R = 1,21312,252,252,252
BEGIN DESCRIPTION:
Mapping XS 60fcf193
END DESCRIPTION:
XS GIS Cut Line= 4
      2828378.23      7013837.61      2828666.41      7013667.48
      2828871.27      7013323.73      2829013.41      7012949.32
#Sta/Elev= 30
  4642.5  462.71  4833.6  460.90  4928.1  458.37  4933.9  458.69  4955.1  456.93
  4997.6  453.41  4998.1  452.61  5003.1  452.61  5003.6  453.41  5006.4  454.57
  5012.0  454.77  5037.6  455.46  5053.0  456.93  5080.4  458.20  5101.8  458.17
  5166.3  460.25  5372.4  464.59  5482.0  464.02  5525.7  462.52  5579.2  462.10
  5589.9  461.80  5602.5  460.73  5643.4  460.27  5687.6  461.29  5696.9  461.07
  5707.0  461.85  5712.4  461.37  5737.2  461.60  5761.0  462.14  5777.8  463.28
#Mann=5,-1,0
  4642.5    0.05       0  4833.6    0.16       0  4997.6    0.07       0
  5003.6    0.16       0  5012.0    0.05       0
Bank Sta=4955.1,5053
Exp/Cntr=0.3,0.1

Type RM Length L Ch R = 1,21060,333,333,333
BEGIN DESCRIPTION:
Mapping XS eb6cf5df
END DESCRIPTION:
XS GIS Cut Line= 3
      2828794.89      7014111.89      2828881.69      7013778.59
      2829013.63      7013032.08
#Sta/Elev= 30
  4654.1  461.11  4774.9  458.93  4832.4  456.82  4872.9  456.99  4880.2  456.40
  4916.0  454.91  4948.8  453.02  4994.4  452.95  4994.8  452.15  4995.3  451.35
  5000.3  451.35  5000.8  452.15  5049.7  454.91  5063.1  456.04  5101.5  457.61
  5144.3  457.70  5387.0  462.35  5446.2  463.22  5451.3  462.85  5479.4  463.00
  5489.6  463.48  5520.1  462.57  5559.5  463.06  5570.8  462.20  5618.7  462.11
  5662.2  460.17  5713.0  459.51  5732.0  459.61  5743.5  460.46  5756.6  460.63
#Mann=5,-1,0
  4654.1    0.05       0  4880.2    0.16       0  4994.8    0.07       0
  5000.8    0.16       0  5101.5    0.05       0
Bank Sta=4916,5049.7
Exp/Cntr=0.3,0.1

Type RM Length L Ch R = 1,20727,173,173,173
BEGIN DESCRIPTION:
Penson Spring Branch 39.0
END DESCRIPTION:
XS GIS Cut Line= 3
      2828974.98      7014075.04      2829175.00      7013675.00
      2828975.01      7013425.02
#Sta/Elev= 30
  4553.0  462.31  4740.3  457.28  4790.6  456.59  4828.5  455.22  4835.4  455.22
  4867.2  452.79  4874.5  452.17  4896.8  451.70  4902.4  451.95  4919.2  451.14
  4941.6  450.85  4947.2  451.59  4955.5  451.24  4963.9  450.25  4969.5  451.00
  4983.3  449.36  4983.8  448.56  4988.8  448.56  4989.3  449.36  4991.9  450.12
  5003.5  449.95  5013.9  450.76  5028.3  450.57  5050.7  451.65  5091.5  452.79
  5117.8  456.20  5149.9  457.40  5156.3  458.19  5220.4  458.82  5320.4  461.32
#Mann=5,-1,0
  4553.0    0.05       0  4828.5    0.16       0  4983.3    0.07       0
  4989.3    0.16       0  5117.8    0.05       0
Bank Sta=4867.2,5091.5
Exp/Cntr=0.3,0.1

Type RM Length L Ch R = 1,20554,227,227,227
BEGIN DESCRIPTION:
Penson Spring Branch 38.0
END DESCRIPTION:
XS GIS Cut Line= 3
      2829218.49      7014076.37      2829338.29      7013623.21
      2829175.01      7013325.01
#Sta/Elev= 30
  4519.4  457.91  4655.3  455.38  4776.5  453.85  4810.4  452.63  4831.1  452.89
  4842.5  453.59  4862.2  453.47  4896.7  451.96  4944.9  451.04  4994.5  448.26
  4995.0  447.46  5000.0  447.46  5000.5  448.26  5004.3  449.37  5020.3  449.30
  5026.1  449.84  5031.8  449.39  5047.9  450.14  5054.5  451.38  5069.7  451.49
  5072.3  451.96  5085.8  455.03  5091.5  454.36  5107.6  456.00  5122.9  455.62
  5145.6  453.33  5156.6  454.13  5189.2  454.70  5216.7  456.16  5328.1  458.62
#Mann=5,-1,0
  4519.4    0.05       0  4776.5    0.16       0  4994.5    0.07       0
  5000.5    0.16       0  5156.6    0.05       0
Bank Sta=4896.7,5072.3
Exp/Cntr=0.3,0.1

Type RM Length L Ch R = 1,20327,297,297,297
BEGIN DESCRIPTION:
Mapping XS 2768c016
END DESCRIPTION:
XS GIS Cut Line= 3
      2829338.30      7014084.12      2829544.02      7013662.27
      2829533.60      7013323.76
#Sta/Elev= 30
  4510.1  455.66  4536.9  455.51  4598.1  453.59  4622.4  454.28  4627.0  454.73
  4664.9  453.15  4687.1  451.08  4700.2  450.87  4722.7  451.52  4739.7  453.84
  4745.2  453.05  4790.3  452.73  4807.3  453.45  4942.5  450.07  4961.6  448.78
  4993.7  447.36  4994.2  446.56  4999.2  446.56  4999.7  447.36  5016.7  448.11
  5076.8  447.63  5086.8  447.84  5092.2  448.78  5105.9  451.66  5110.9  450.30
  5116.8  452.77  5122.8  453.37  5156.8  454.82  5226.8  453.89  5318.1  455.83
#Mann=5,-1,0
  4510.1    0.05       0  4622.4    0.16       0  4993.7    0.07       0
  4999.7    0.16       0  5122.8    0.05       0
Bank Sta=4961.6,5092.2
Exp/Cntr=0.3,0.1

Type RM Length L Ch R = 1,20030,288,288,288
BEGIN DESCRIPTION:
Mapping XS b41825c1
END DESCRIPTION:
XS GIS Cut Line= 4
      2829658.59      7014170.11      2829783.60      7013795.08
      2829799.22      7013657.06      2829783.67      7013348.57
#Sta/Elev= 30
  4588.2  457.15  4677.9  455.48  4685.4  455.52  4690.6  456.10  4748.6  454.38
  4836.0  453.16  4867.7  452.24  4899.3  450.49  4920.4  447.87  4940.8  446.62
  4962.5  445.64  4975.2  445.62  4980.9  444.69  4986.1  444.69  4990.7  443.60
  4991.2  442.80  4996.2  442.80  4996.7  443.60  5014.2  444.85  5033.9  445.58
  5042.6  446.62  5064.1  448.34  5094.3  449.56  5114.4  449.85  5142.4  449.39
  5194.6  451.06  5204.6  450.92  5244.6  452.03  5324.7  452.40  5431.3  453.94
#Mann=5,-1,0
  4588.2    0.05       0  4990.7    0.03       0  4996.7    0.05       0
  5014.2    0.16       0  5142.4    0.05       0
Bank Sta=4940.8,5042.6
Exp/Cntr=0.3,0.1

Type RM Length L Ch R = 1,19742,508,508,508
BEGIN DESCRIPTION:
Penson Spring Branch 37.0
END DESCRIPTION:
XS GIS Cut Line= 3
      2830025.00      7013975.03      2830040.32      7013748.47
      2829975.00      7013375.01
#Sta/Elev= 30
  4774.5  451.81  4849.2  449.98  4925.5  445.56  4929.4  445.40  4954.9  443.88
  4965.0  443.56  4975.0  443.30  4998.4  443.91  5000.8  443.54  5006.8  443.72
  5012.2  442.86  5012.7  442.06  5017.7  442.06  5018.2  442.86  5025.4  443.85
  5039.7  443.78  5061.2  444.89  5087.0  445.56  5137.1  447.53  5157.4  449.30
  5180.2  449.72  5218.3  448.25  5248.7  448.37  5279.2  449.13  5289.0  450.00
  5294.0  449.96  5299.5  450.95  5309.7  451.52  5353.5  452.28  5380.7  452.30
#Mann=5,-1,0
  4774.5    0.05       0  4929.4    0.16       0  5012.2    0.07       0
  5018.2    0.16       0  5039.7    0.05       0
Bank Sta=4925.5,5087
Exp/Cntr=0.3,0.1

Type RM Length L Ch R = 1,19234,88,88,88
BEGIN DESCRIPTION:
Penson Spring Branch 36.0
END DESCRIPTION:
XS GIS Cut Line= 3
      2830491.94      7013956.56      2830445.06      7013716.96
      2830447.66      7013250.81
#Sta/Elev= 30
  4623.4  451.19  4683.3  449.65  4688.4  450.05  4692.4  449.84  4786.3  446.04
  4791.4  446.32  4837.8  444.26  4842.9  444.44  4858.3  441.98  4866.0  440.80
  4879.5  440.44  4899.5  440.87  4919.5  440.50  4939.5  440.87  4989.5  440.75
  4996.5  438.20  4997.0  437.40  5002.0  437.40  5002.5  438.20  5009.5  439.85
  5019.5  440.67  5049.5  441.10  5060.5  441.98  5079.5  444.41  5099.5  445.18
  5149.5  444.96  5193.8  445.31  5219.5  445.24  5249.5  445.83  5333.7  448.39
#Mann=5,-1,0
  4623.4    0.08       0  4692.4    0.16       0  4996.5    0.07       0
  5002.5    0.16       0  5193.8    0.05       0
Bank Sta=4858.3,5060.5
Exp/Cntr=0.3,0.1

Type RM Length L Ch R = 1,19146,217,217,217
BEGIN DESCRIPTION:
Mapping XS 127b82db
END DESCRIPTION:
XS GIS Cut Line= 3
      2830583.08      7013953.94      2830533.60      7013758.62
      2830533.60      7013279.71
#Sta/Elev= 30
  4631.2  449.83  4656.8  449.52  4671.4  449.52  4680.5  448.87  4685.6  449.02
  4692.0  448.14  4767.6  446.11  4775.4  445.24  4803.5  444.28  4815.8  444.73
  4832.0  443.30  4875.4  441.58  4906.3  440.54  4976.3  440.36  4986.4  439.95
  5013.3  437.46  5013.8  436.66  5018.8  436.66  5019.3  437.46  5026.3  439.57
  5030.3  439.95  5036.3  440.51  5066.3  440.96  5086.3  442.70  5106.3  443.51
  5168.9  442.83  5186.3  443.61  5236.3  443.80  5266.7  445.19  5311.6  448.34
#Mann=8,-1,0
  4631.2    0.05       0  4656.8    0.08       0  4775.4    0.05       0
  4875.4    0.08       0  5013.3    0.07       0  5019.3    0.08       0
  5168.9    0.05       0  5266.7    0.08       0
Bank Sta=4986.4,5030.3
Exp/Cntr=0.3,0.1

Type RM Length L Ch R = 1,18929,280,280,280
BEGIN DESCRIPTION:
Penson Spring Branch 35.0
END DESCRIPTION:
XS GIS Cut Line= 3
      2830624.99      7013975.03      2830725.00      7013675.00
      2830675.00      7013374.99
#Sta/Elev= 30
  4680.7  450.46  4701.8  448.97  4754.5  447.86  4796.7  445.38  4817.8  444.76
  4849.4  441.78  4881.0  440.79  4912.6  438.58  4923.2  437.26  4933.6  437.01
  4965.3  437.51  4975.9  436.76  4983.4  433.59  4983.9  432.79  4988.9  432.79
  4989.4  433.59  4999.5  433.62  5007.1  434.43  5024.8  437.48  5029.9  435.03
  5037.5  435.39  5046.8  437.01  5067.9  438.18  5118.6  439.20  5146.5  441.72
  5151.6  441.23  5169.3  444.02  5189.6  445.54  5268.1  446.39  5301.1  447.48
#Mann=3,-1,0
  4680.7    0.05       0  4983.4    0.03       0  4989.4    0.05       0
Bank Sta=4933.6,5046.8
Exp/Cntr=0.3,0.1

Type RM Length L Ch R = 1,18649,185,185,185
BEGIN DESCRIPTION:
Penson Spring Branch 34.0
END DESCRIPTION:
XS GIS Cut Line= 3
      2830724.97      7014125.03      2830925.00      7013875.00
      2830974.99      7013575.03
#Sta/Elev= 30
  4665.8  452.08  4673.0  451.99  4772.3  447.54  4793.9  445.65  4844.3  443.22
  4865.1  441.53  4885.9  440.80  4943.6  437.44  4950.0  437.57  4958.0  437.02
  4964.4  437.17  4972.4  436.61  4978.8  436.59  4980.0  435.61  4982.8  433.29
  4988.5  433.29  4993.1  432.34  4993.6  431.54  4998.6  431.54  4999.1  432.34
  5006.3  434.96  5013.9  435.92  5046.8  435.40  5055.1  435.61  5079.8  436.30
  5087.4  437.09  5107.7  437.36  5148.2  439.91  5219.2  443.59  5290.1  446.14
#Mann=3,-1,0
  4665.8    0.05       0  4993.1    0.03       0  4999.1    0.05       0
Bank Sta=4980,5055.1
Exp/Cntr=0.3,0.1

Type RM Length L Ch R = 1,18464,155,155,155
BEGIN DESCRIPTION:
Mapping XS 875faa04
END DESCRIPTION:
XS GIS Cut Line= 3
      2830950.28      7014149.22      2831089.96      7013939.85
      2831118.23      7013708.15
#Sta/Elev= 30
  4753.2  447.69  4803.5  445.98  4818.4  446.06  4830.6  445.57  4839.6  444.32
  4860.6  442.56  4911.7  438.84  4947.8  436.75  4953.8  436.01  4974.8  435.44
  4983.7  434.45  4989.8  433.15  4998.7  432.56  5001.8  431.73  5002.3  430.93
  5007.3  430.93  5007.8  431.73  5029.9  435.01  5080.3  434.95  5110.5  434.21
  5119.9  434.45  5140.7  435.03  5168.1  437.53  5173.2  436.55  5191.1  438.35
  5201.2  440.00  5211.3  442.41  5221.3  445.47  5231.4  447.53  5238.3  447.68
#Mann=3,-1,0
  4753.2    0.05       0  5001.8    0.03       0  5007.8    0.05       0
Bank Sta=4983.7,5119.9
Exp/Cntr=0.3,0.1

Type RM Length L Ch R = 1,18309,346,346,346
BEGIN DESCRIPTION:
Penson Spring Branch 33.0
END DESCRIPTION:
XS GIS Cut Line= 3
      2830974.99      7014225.01      2831225.00      7014025.00
      2831424.99      7013775.02
#Sta/Elev= 30
  4710.6  448.65  4767.4  447.20  4781.8  447.45  4802.7  446.11  4810.7  445.00
  4825.1  445.13  4874.7  442.66  4938.7  436.99  4945.1  437.08  4953.1  435.66
  4959.5  435.81  4966.7  434.38  4981.2  432.68  4988.3  429.99  4991.7  428.17
  4992.2  427.37  4997.2  427.37  4997.7  428.17  5002.8  432.48  5003.9  432.68
  5009.2  433.64  5081.2  433.23  5144.0  436.79  5170.1  438.85  5230.1  442.20
  5258.9  444.79  5286.9  446.66  5314.9  447.44  5322.9  448.74  5350.9  449.35
#Mann=5,-1,0
  4710.6    0.05       0  4991.7    0.03       0  4997.7    0.05       0
  5144.0    0.16       0  5170.1    0.05       0
Bank Sta=4981.2,5003.9
Exp/Cntr=0.3,0.1

Type RM Length L Ch R = 1,17963,378,378,378
BEGIN DESCRIPTION:
Penson Spring Branch 32.0
END DESCRIPTION:
XS GIS Cut Line= 3
      2831075.01      7014275.00      2831375.00      7014325.00
      2831524.98      7014025.03
#Sta/Elev= 30
  4689.2  446.08  4722.1  441.64  4846.2  435.63  4899.4  431.90  4932.5  431.14
  4952.8  429.48  4960.4  429.37  4965.4  431.03  4973.1  430.51  4980.2  426.10
  4980.7  425.30  4985.7  425.30  4986.2  426.10  4996.1  426.71  5001.7  430.66
  5007.3  429.64  5033.9  431.66  5042.9  431.90  5046.4  432.02  5052.0  434.42
  5068.8  434.01  5074.4  435.79  5119.1  438.62  5135.9  438.31  5180.6  439.93
  5186.2  441.07  5247.7  441.43  5253.3  442.38  5292.4  443.87  5328.7  444.42
#Mann=5,-1,0
  4689.2    0.05       0  4846.2    0.16       0  4980.2    0.07       0
  4986.2    0.16       0  5033.9    0.05       0
Bank Sta=4899.4,5042.9
Exp/Cntr=0.3,0.1

Type RM Length L Ch R = 1,17585,329,329,329
BEGIN DESCRIPTION:
Penson Spring Branch 31.0
END DESCRIPTION:
XS GIS Cut Line= 3
      2831425.03      7014774.97      2831625.00      7014525.00
      2831625.00      7014225.01
#Sta/Elev= 30
  4672.9  443.68  4729.7  441.03  4744.1  439.59  4827.2  434.90  4851.3  433.02
  4857.7  432.99  4886.6  429.62  4894.8  429.48  4901.0  428.86  4907.4  429.62
  4915.4  428.21  4921.8  428.49  4942.6  427.25  4957.0  428.56  4971.4  428.50
  4979.4  429.18  4985.8  428.70  4986.8  424.88  4987.3  424.08  4992.3  424.08
  4992.8  424.88  4995.5  424.88  5003.0  427.54  5013.0  429.03  5045.7  429.48
  5073.0  430.78  5107.6  433.51  5213.0  441.12  5283.0  443.46  5293.0  443.45
#Mann=5,-1,0
  4672.9    0.05       0  4827.2    0.16       0  4986.8    0.07       0
  4992.8    0.16       0  5107.6    0.05       0
Bank Sta=4894.8,5045.7
Exp/Cntr=0.3,0.1

Type RM Length L Ch R = 1,17256,487,487,487
BEGIN DESCRIPTION:
Penson Spring Branch 30.0
END DESCRIPTION:
XS GIS Cut Line= 3
      2831824.99      7014925.05      2831875.00      7014625.00
      2831725.00      7014325.00
#Sta/Elev= 30
  4737.7  440.95  4758.0  440.89  4831.5  439.37  4859.4  438.06  4940.0  431.69
  4948.1  430.52  4953.2  430.79  4973.5  427.51  4981.1  426.28  4988.2  421.92
  4988.7  421.12  4993.7  421.12  4994.2  421.92  5001.3  424.21  5008.9  425.46
  5014.0  422.25  5021.6  422.34  5031.7  426.74  5050.3  426.91  5063.2  427.51
  5149.1  428.64  5212.4  429.61  5259.8  432.03  5301.8  435.08  5318.6  436.99
  5324.2  437.19  5341.0  439.44  5363.3  441.15  5368.9  440.51  5377.3  441.29
#Mann=6,-1,0
  4737.7    0.05       0  4940.0    0.16       0  4988.2    0.07       0
  4994.2    0.16       0  5149.1    0.12       0  5259.8    0.05       0
Bank Sta=4973.5,5063.2
Exp/Cntr=0.3,0.1

Type RM Length L Ch R = 1,16769,408,408,408
BEGIN DESCRIPTION:
Penson Spring Branch 29.0
END DESCRIPTION:
XS GIS Cut Line= 3
      2832113.15      7014979.82      2832175.00      7014625.00
      2832125.00      7014325.01
#Sta/Elev= 30
  4619.3  432.74  4696.5  431.70  4713.9  431.32  4725.7  430.48  4766.3  429.86
  4806.9  428.32  4827.9  426.96  4838.2  426.21  4847.5  426.49  4892.7  425.39
  4938.9  425.79  4947.1  425.40  4969.2  425.46  4982.0  425.29  4989.6  424.21
  4996.7  421.27  4997.2  420.47  5002.2  420.47  5002.7  421.27  5007.4  421.57
  5012.4  424.13  5020.0  425.86  5031.2  426.96  5040.3  427.91  5068.2  428.18
  5162.0  433.29  5182.2  433.43  5202.5  434.84  5222.8  435.46  5283.6  439.23
#Mann=5,-1,0
  4619.3    0.05       0  4696.5    0.16       0  4969.2    0.05       0
  4996.7    0.03       0  5002.7    0.05       0
Bank Sta=4827.9,5031.2
Exp/Cntr=0.3,0.1

Type RM Length L Ch R = 1,16361,400,400,400
BEGIN DESCRIPTION:
Penson Spring Branch 28.0
END DESCRIPTION:
XS GIS Cut Line= 3
      2832075.04      7015124.97      2832375.00      7014875.00
      2832624.98      7014675.01
#Sta/Elev= 30
  4639.4  437.82  4717.5  431.71  4785.4  429.77  4823.5  428.15  4831.4  427.26
  4871.7  426.30  4895.1  424.66  4916.0  425.32  4944.6  424.98  4958.9  422.89
  4979.7  423.80  4994.1  423.55  4998.9  418.33  4999.4  417.53  5004.4  417.53
  5004.9  418.33  5016.2  422.16  5022.7  423.40  5033.1  423.62  5037.1  424.96
  5053.7  426.30  5072.3  427.54  5115.5  432.75  5130.4  433.69  5165.1  437.14
  5193.9  438.99  5222.0  439.56  5243.6  439.07  5286.0  439.64  5350.0  439.48
#Mann=5,-1,0
  4639.4    0.05       0  4785.4    0.16       0  4998.9    0.07       0
  5004.9    0.16       0  5130.4    0.05       0
Bank Sta=4871.7,5053.7
Exp/Cntr=0.3,0.1

Type RM Length L Ch R = 1,15961,356,356,356
BEGIN DESCRIPTION:
Penson Spring Branch 27.0
END DESCRIPTION:
XS GIS Cut Line= 3
      2832174.98      7015275.01      2832525.00      7015125.00
      2832624.99      7014825.03
#Sta/Elev= 30
  4592.3  437.63  4712.0  428.51  4776.5  424.73  4813.2  422.82  4829.9  421.92
  4864.3  424.07  4884.5  423.85  4906.0  422.95  4940.5  423.07  4958.6  421.20
  4964.0  422.45  4983.6  421.95  4994.2  418.00  5001.7  417.04  5002.2  416.24
  5007.2  416.24  5007.7  417.04  5015.3  422.20  5019.4  422.82  5025.8  423.80
  5046.9  424.68  5057.4  426.41  5078.5  428.34  5089.1  430.76  5112.3  432.34
  5120.7  433.82  5141.8  434.95  5152.3  436.26  5215.5  438.24  5289.3  438.87
#Mann=6,-1,0
  4592.3    0.16       0  4776.5    0.12       0  4884.5    0.16       0
  5001.7    0.07       0  5007.7    0.16       0  5112.3    0.05       0
Bank Sta=4813.2,5019.4
Exp/Cntr=0.3,0.1

Type RM Length L Ch R = 1,15605,119,119,119
BEGIN DESCRIPTION:
Mapping XS 0fd09556
END DESCRIPTION:
XS GIS Cut Line= 3
      2832235.73      7015350.90      2832607.30      7015357.84
      2833081.47      7015371.69
#Sta/Elev= 30
  4640.8  435.86  4643.0  435.86  4660.1  433.80  4731.3  428.35  4750.1  427.12
  4789.4  425.38  4830.1  422.63  4864.5  421.98  4890.1  421.67  4929.3  422.20
  4950.1  421.17  4970.1  421.59  4980.1  421.34  4990.1  419.53  4997.1  416.00
  4997.6  415.20  5002.6  415.20  5003.1  416.00  5008.8  417.81  5012.4  417.81
  5020.1  421.35  5028.3  421.12  5120.2  420.41  5140.2  421.20  5200.2  421.96
  5230.2  421.04  5290.3  420.64  5427.1  422.45  5433.3  421.98  5486.8  423.58
#Mann=7,-1,0
  4640.8    0.05       0  4731.3    0.16       0  4789.4    0.12       0
  4929.3    0.07       0  4997.1    0.07       0  5003.1    0.07       0
  5028.3    0.05       0
Bank Sta=4864.5,5433.3
Exp/Cntr=0.3,0.1

Type RM Length L Ch R = 1,15486,878,878,878
BEGIN DESCRIPTION:
Mapping XS 73981e27
END DESCRIPTION:
XS GIS Cut Line= 5
      2832350.34      7015555.77      2832461.46      7015472.43
      2833010.07      7015448.12      2833096.88      7015448.12
      2833120.58      7015377.02
#Sta/Elev= 30
  4682.8  429.26  4772.8  427.46  4875.4  421.77  4915.3  420.39  4965.4  421.39
  4975.4  420.24  4982.4  415.21  4982.9  414.41  4987.9  414.41  4988.4  415.21
  5005.0  420.52  5025.4  421.40  5055.5  420.83  5065.5  421.48  5095.5  420.54
  5106.5  421.35  5125.5  420.79  5185.6  421.37  5215.6  420.45  5255.7  421.28
  5385.8  419.28  5461.9  419.64  5466.6  420.31  5472.1  420.48  5477.6  421.77
  5482.0  422.82  5492.6  423.33  5498.5  422.32  5513.7  422.96  5532.6  425.09
#Mann=5,-1,0
  4682.8    0.16       0  4982.4    0.07       0  4988.4    0.16       0
  5005.0    0.12       0  5466.6    0.05       0
Bank Sta=4875.4,5477.6
Exp/Cntr=0.3,0.1

Type RM Length L Ch R = 1,14608,282,282,282
BEGIN DESCRIPTION:
Penson Spring Branch 24.0
END DESCRIPTION:
XS GIS Cut Line= 3
      2833125.00      7016025.01      2833175.00      7015675.00
      2833175.00      7015274.97
#Sta/Elev= 30
  4515.3  436.04  4656.7  427.99  4737.5  424.22  4808.5  420.31  4836.0  419.44
  4878.9  419.43  4888.9  419.09  4898.9  416.08  4908.9  415.45  4928.9  416.68
  4938.9  418.89  4968.9  418.15  4978.9  417.39  4988.9  415.07  4995.9  411.79
  4996.4  410.99  5001.4  410.99  5001.9  411.79  5008.9  416.61  5018.9  418.67
  5028.9  418.10  5048.9  417.96  5085.8  419.44  5098.9  419.92  5102.5  420.53
  5118.9  423.40  5138.9  422.64  5158.9  424.91  5218.9  430.53  5268.9  434.56
#Mann=5,-1,0
  4515.3    0.16       0  4808.5    0.12       0  4995.9    0.07       0
  5001.9    0.12       0  5102.5    0.05       0
Bank Sta=4836,5085.8
Exp/Cntr=0.3,0.1

Type RM Length L Ch R = 1,14326,66,66,66
BEGIN DESCRIPTION:
Mapping XS 6dec72a1
END DESCRIPTION:
XS GIS Cut Line= 3
      2833318.24      7016029.68      2833349.48      7015501.07
      2833318.24      7015204.24
#Sta/Elev= 30
  4473.2  435.52  4518.0  434.05  4568.9  433.45  4618.1  432.06  4667.9  427.83
  4678.2  425.99  4718.3  422.11  4738.3  421.11  4868.6  418.69  4918.7  418.98
  4968.7  417.71  4978.8  412.55  4985.8  412.13  4986.3  411.33  4991.3  411.33
  4991.8  412.13  4998.3  415.80  5002.7  415.80  5008.8  416.99  5018.9  416.20
  5028.9  417.91  5040.8  418.69  5069.2  420.94  5119.4  419.91  5157.4  421.98
  5186.8  423.61  5199.9  425.17  5279.8  427.89  5286.8  428.88  5301.2  429.76
#Mann=6,-1,0
  4473.2    0.08       0  4568.9    0.05       0  4985.8    0.04       0
  4991.8    0.05       0  5157.4    0.08       0  5286.8    0.05       0
Bank Sta=4868.6,5040.8
Exp/Cntr=0.3,0.1

Type RM Length L Ch R = 1,14260,464,464,464
BEGIN DESCRIPTION:
Mapping XS 359292cb
END DESCRIPTION:
XS GIS Cut Line= 3
      2833406.78      7015990.62      2833414.59      7015498.47
      2833440.63      7015045.33
#Sta/Elev= 30
  4509.0  432.45  4544.6  431.80  4565.7  429.12  4584.6  430.77  4604.6  430.34
  4644.6  428.55  4659.5  426.09  4664.6  425.00  4684.6  425.14  4694.6  424.43
  4724.6  420.85  4734.7  420.39  4855.6  418.83  4885.4  418.60  4924.7  418.68
  4974.7  416.68  4991.7  410.89  4992.2  410.09  4997.2  410.09  4997.7  410.89
  5014.7  412.07  5024.7  415.89  5034.7  417.41  5099.4  418.60  5225.1  421.51
  5270.0  420.63  5385.3  421.98  5405.4  423.41  5435.6  424.16  5455.1  424.07
#Mann=7,-1,0
  4509.0    0.16       0  4565.7    0.05       0  4659.5    0.16       0
  4855.6    0.12       0  4991.7    0.07       0  4997.7    0.12       0
  5435.6    0.16       0
Bank Sta=4885.4,5099.4
Exp/Cntr=0.3,0.1

Type RM Length L Ch R = 1,13796,537,537,537
BEGIN DESCRIPTION:
Penson Spring Branch 22.0
END DESCRIPTION:
XS GIS Cut Line= 3
      2833424.98      7015975.01      2833725.00      7015775.00
      2833875.01      7015374.98
#Sta/Elev= 30
  4614.9  431.03  4643.5  429.64  4673.5  426.90  4679.5  427.98  4715.6  427.61
  4736.6  424.71  4759.1  423.81  4781.7  421.32  4872.4  417.36  4931.9  415.97
  4973.2  416.79  4985.3  416.17  4990.6  414.16  4993.8  409.63  4994.3  408.83
  4999.3  408.83  4999.8  409.63  5007.5  415.97  5015.5  416.22  5070.7  416.19
  5106.3  415.12  5211.4  416.06  5241.6  414.73  5246.9  416.06  5249.1  417.36
  5253.2  419.74  5271.8  423.66  5277.2  423.45  5315.0  428.22  5402.7  435.40
#Mann=6,-1,0
  4614.9    0.16       0  4973.2    0.12       0  4993.8    0.07       0
  4999.8    0.12       0  5211.4    0.16       0  5315.0    0.05       0
Bank Sta=4872.4,5249.1
Exp/Cntr=0.3,0.1

Type RM Length L Ch R = 1,13259,586,586,586
BEGIN DESCRIPTION:
Penson Spring Branch 21.0
END DESCRIPTION:
XS GIS Cut Line= 3
      2833824.98      7016375.02      2834125.00      7016025.00
      2834175.00      7015574.97
#Sta/Elev= 30
  4531.6  433.79  4716.0  429.92  4723.2  428.32  4729.7  428.44  4737.4  426.98
  4744.0  427.17  4845.8  417.86  4869.5  415.61  4928.4  413.48  4985.5  414.53
  4989.3  413.21  4995.1  413.21  5002.7  408.65  5009.7  407.72  5010.2  406.92
  5015.3  406.92  5015.8  407.72  5022.8  411.85  5032.9  414.22  5123.4  415.54
  5163.1  415.28  5171.2  415.61  5234.1  418.38  5261.3  421.07  5294.5  426.41
  5335.7  427.13  5364.9  428.28  5395.1  431.05  5405.1  432.81  5445.4  433.54
#Mann=7,-1,0
  4531.6    0.05       0  4845.8    0.16       0  5009.7    0.07       0
  5015.8    0.16       0  5163.1    0.05       0  5261.3    0.16       0
  5335.7    0.05       0
Bank Sta=4869.5,5171.2
Exp/Cntr=0.3,0.1

Type RM Length L Ch R = 1,12673,496,496,496
BEGIN DESCRIPTION:
Penson Spring Branch 20.0
END DESCRIPTION:
XS GIS Cut Line= 3
      2834225.00      7016525.00      2834575.00      7016225.00
      2834725.00      7015775.01
#Sta/Elev= 30
  4521.3  431.49  4569.8  429.50  4599.8  426.89  4620.6  423.67  4649.2  420.80
  4663.4  419.58  4670.0  420.07  4677.7  418.07  4700.6  415.88  4757.4  413.38
  4819.3  411.45  4882.9  413.39  4975.1  411.77  4984.9  412.22  4992.8  408.40
  5000.3  406.59  5000.8  405.79  5005.9  405.79  5006.4  406.59  5013.9  411.81
  5108.8  411.86  5118.8  413.38  5129.8  416.58  5161.5  422.11  5182.6  423.88
  5193.1  425.75  5255.7  429.72  5288.0  431.07  5348.8  431.48  5456.6  431.81
#Mann=7,-1,0
  4521.3    0.05       0  4569.8    0.16       0  4700.6    0.12       0
  5000.3    0.07       0  5006.4    0.12       0  5255.7    0.16       0
  5348.8    0.05       0
Bank Sta=4757.4,5118.8
Exp/Cntr=0.3,0.1

Type RM Length L Ch R = 1,12177,568,568,568
BEGIN DESCRIPTION:
Mapping XS c9ba0231
END DESCRIPTION:
XS GIS Cut Line= 3
      2834532.65      7016826.59      2834810.42      7016362.18
      2834849.19      7016108.06
#Sta/Elev= 30
  4407.9  428.22  4424.7  427.25  4440.3  425.23  4461.7  424.14  4584.5  414.26
  4650.3  413.03  4696.0  411.89  4737.9  410.38  4769.0  410.95  4805.9  410.11
  4827.4  410.70  4864.2  410.23  4976.5  411.02  4986.7  410.52  4993.7  404.95
  4994.2  404.15  4999.4  404.15  4999.9  404.95  5006.9  405.83  5012.2  410.65
  5037.2  410.36  5057.5  409.25  5066.0  411.89  5075.8  416.08  5080.8  416.41
  5087.8  419.46  5097.9  421.70  5142.6  427.04  5168.7  429.03  5206.1  429.61
#Mann=5,-1,0
  4407.9    0.16       0  4650.3    0.12       0  4993.7    0.07       0
  4999.9    0.12       0  5142.6    0.16       0
Bank Sta=4696,5066
Exp/Cntr=0.3,0.1

Type RM Length L Ch R = 1,11609,623,623,623
BEGIN DESCRIPTION:
Mapping XS b3c73512
END DESCRIPTION:
XS GIS Cut Line= 3
      2834862.52      7016965.45      2834992.71      7016531.45
      2834975.35      7016231.96
#Sta/Elev= 30
  4504.4  424.00  4508.1  423.97  4536.2  420.46  4623.2  415.03  4742.3  410.80
  4758.5  410.57  4800.9  409.24  4810.9  409.23  4818.1  405.03  4828.5  406.61
  4838.7  409.92  4870.3  410.30  4891.2  408.64  4910.0  409.43  4915.3  405.89
  4922.5  408.45  4948.3  408.34  4974.0  409.89  4984.0  408.78  4998.6  403.47
  4999.1  402.67  5004.8  403.47  5006.7  407.93  5014.1  409.10  5084.2  410.15
  5114.2  408.88  5136.7  410.57  5194.4  413.73  5214.4  418.31  5257.5  422.45
#Mann=7,-1,0
  4504.4    0.16       0  4508.1    0.05       0  4623.2    0.12       0
  4742.3    0.16       0  4800.9    0.12       0  4998.6    0.07       0
  5004.8    0.12       0
Bank Sta=4758.5,5136.7
Exp/Cntr=0.3,0.1

Type RM Length L Ch R = 1,10986,684,684,684
BEGIN DESCRIPTION:
Penson Spring Branch 19.0
END DESCRIPTION:
XS GIS Cut Line= 3
      2835283.51      7016978.50      2835325.00      7016625.00
      2835313.93      7016038.33
#Sta/Elev= 30
  4631.0  417.65  4654.7  418.27  4674.8  417.16  4683.2  417.81  4688.3  416.90
  4705.0  419.40  4725.1  419.48  4779.3  417.86  4846.0  417.19  4906.4  415.29
  4942.8  410.80  4947.9  411.29  4966.7  408.76  4974.3  406.70  4976.9  405.99
  4981.3  402.55  4981.8  401.75  4987.0  401.75  4987.5  402.55  4996.9  403.07
  5006.9  406.71  5016.9  408.15  5237.0  406.99  5246.9  408.05  5319.3  408.76
  5356.3  409.52  5367.0  409.33  5417.0  412.20  5507.0  418.52  5573.7  422.08
#Mann=6,-1,0
  4631.0    0.05       0  4779.3    0.16       0  4974.3    0.12       0
  4981.3    0.07       0  4987.5    0.12       0  5356.3    0.16       0
Bank Sta=4966.7,5319.3
Exp/Cntr=0.3,0.1

Type RM Length L Ch R = 1,10302,660,660,660
BEGIN DESCRIPTION:
Penson Spring Branch 18.0
END DESCRIPTION:
XS GIS Cut Line= 3
      2835474.98      7017075.03      2835725.00      7016525.00
      2836075.02      7016224.98
#Sta/Elev= 30
  4333.9  424.77  4365.8  423.82  4446.0  417.12  4535.8  412.50  4589.9  409.58
  4687.6  408.07  4710.7  407.70  4740.4  408.74  4774.3  407.39  4808.5  406.31
  4828.3  402.69  4828.8  401.89  4834.3  401.89  4834.8  402.69  4854.6  405.66
  4933.3  406.55  4951.8  405.42  4959.5  403.11  4966.1  405.67  4973.8  402.90
  4980.3  404.82  4994.6  402.86  5008.9  403.92  5016.6  406.59  5039.5  407.39
  5122.5  411.44  5158.2  414.02  5242.7  422.01  5320.6  427.15  5399.1  429.17
#Mann=6,-1,0
  4333.9    0.05       0  4535.8    0.16       0  4687.6    0.12       0
  4828.3    0.03       0  4834.8    0.12       0  4933.3    0.05       0
Bank Sta=4774.3,5039.5
Exp/Cntr=0.3,0.1

Type RM Length L Ch R = 1,9642,98,98,98
BEGIN DESCRIPTION:
Mapping XS 214b74b1
END DESCRIPTION:
XS GIS Cut Line= 4
      2835905.05      7017357.82      2836033.51      7017135.62
      2836043.93      7016934.23      2836050.87      7016493.31
#Sta/Elev= 30
  4562.2  420.91  4600.1  418.97  4614.7  417.62  4630.5  417.33  4636.3  416.49
  4657.9  415.43  4695.1  412.05  4748.2  409.44  4754.0  408.75  4849.7  405.85
  4886.6  404.96  4929.6  404.56  4939.5  404.10  4944.6  403.10  4949.7  402.84
  4959.7  403.91  4976.4  402.49  4976.9  401.69  4982.5  401.69  4983.0  402.49
  5009.7  402.94  5017.6  404.44  5088.1  404.45  5169.8  405.04  5199.5  405.85
  5219.8  406.18  5249.8  408.11  5309.8  410.43  5410.5  416.74  5461.5  419.40
#Mann=6,-1,0
  4562.2    0.05       0  4600.1    0.16       0  4886.6    0.12       0
  4976.4    0.07       0  4983.0    0.12       0  5088.1    0.05       0
Bank Sta=4849.7,5199.5
Exp/Cntr=0.3,0.1

Type RM Length L Ch R = 1,9544,391,391,391
BEGIN DESCRIPTION:
Mapping XS 69b7f9da
END DESCRIPTION:
XS GIS Cut Line= 4
      2836179.34      7017475.88      2836120.32      7017291.87
      2836127.26      7016982.84      2836155.02      7016649.75
#Sta/Elev= 30
  4491.7  421.88  4558.0  418.93  4629.2  414.24  4654.3  413.11  4721.8  409.24
  4741.8  408.44  4785.5  405.48  4811.9  404.35  4831.9  403.99  4900.6  403.75
  4941.9  404.43  4961.9  403.28  4971.9  403.26  4978.6  402.51  4979.1  401.71
  4984.7  401.71  4985.2  402.51  4994.1  402.55  5012.0  403.46  5022.0  403.23
  5032.0  404.43  5042.1  403.58  5096.5  403.71  5142.4  404.26  5181.6  405.48
  5232.7  410.27  5262.8  412.36  5267.8  413.15  5272.9  413.00  5328.3  416.13
#Mann=5,-1,0
  4491.7    0.05       0  4900.6    0.16       0  4978.6    0.07       0
  4985.2    0.16       0  5096.5    0.05       0
Bank Sta=4785.5,5181.6
Exp/Cntr=0.3,0.1

Type RM Length L Ch R = 1,9153,579,579,579
BEGIN DESCRIPTION:
Penson Spring Branch 16.0
END DESCRIPTION:
XS GIS Cut Line= 3
      2836325.00      7017524.99      2836475.00      7017075.00
      2836824.98      7016675.03
#Sta/Elev= 30
  4533.9  424.26  4576.1  423.48  4639.3  420.09  4649.8  418.27  4670.9  417.19
  4702.5  414.22  4713.1  412.35  4776.3  406.75  4808.0  404.68  4869.2  402.46
  4896.0  401.96  4976.6  403.84  4987.1  402.53  4998.3  402.65  5022.0  403.99
  5029.6  402.91  5078.9  401.12  5123.3  401.42  5150.1  401.58  5161.0  399.71
  5161.5  398.91  5167.2  398.91  5167.7  399.71  5178.6  401.59  5234.9  402.46
  5291.5  408.04  5313.4  411.28  5355.1  414.95  5497.5  435.30  5539.7  438.02
#Mann=6,-1,0
  4533.9    0.05       0  4896.0    0.16       0  4998.3     0.1       0
  5123.3    0.05       0  5161.0    0.07       0  5167.7    0.05       0
Bank Sta=4869.2,5234.9
Exp/Cntr=0.3,0.1

Type RM Length L Ch R = 1,8574,450,450,450
BEGIN DESCRIPTION:
Penson Spring Branch 15.0
END DESCRIPTION:
XS GIS Cut Line= 3
      2836925.00      7017775.02      2837025.00      7017125.00
      2836875.00      7016675.01
#Sta/Elev= 30
  4316.0  420.11  4345.1  418.58  4350.2  419.07  4413.4  414.14  4481.7  410.39
  4599.3  402.24  4618.2  401.57  4687.0  399.34  4687.5  398.54  4693.2  398.54
  4693.7  399.34  4791.5  399.34  4862.4  400.55  4892.7  399.36  4933.2  400.25
  4971.1  399.34  5107.0  399.77  5152.9  400.50  5165.5  401.57  5173.9  403.79
  5184.5  404.59  5195.0  406.74  5210.9  408.41  5268.8  413.75  5300.4  418.98
  5332.1  424.94  5342.6  427.54  5395.3  435.39  5416.4  437.24  5448.0  438.32
#Mann=5,-1,0
  4316.0    0.05       0  4687.0   0.033       0  4693.7    0.05       0
  5107.0    0.16       0  5210.9    0.05       0
Bank Sta=4618.2,5165.5
Exp/Cntr=0.3,0.1

Type RM Length L Ch R = 1,8124,178,178,178
BEGIN DESCRIPTION:
Mapping XS 109af196
END DESCRIPTION:
XS GIS Cut Line= 5
      2837550.87      7017854.36      2837467.54      7017614.79
      2837380.73      7017350.90      2837300.87      7017090.48
      2837241.84      7016701.58
#Sta/Elev= 30
  4455.0  418.03  4520.8  417.39  4614.1  413.05  4665.8  407.96  4671.0  408.07
  4696.9  405.10  4719.0  404.02  4727.5  402.87  4759.0  401.37  4771.6  400.37
  4792.1  399.94  4831.3  400.01  4840.5  399.88  4857.5  399.34  4858.0  398.54
  4863.8  398.54  4864.3  399.34  4935.1  399.34  5145.5  399.34  5244.7  399.34
  5304.8  399.44  5419.6  401.37  5426.7  401.64  5456.6  402.42  5497.0  405.47
  5526.8  408.80  5531.8  408.30  5547.6  410.55  5624.0  418.49  5652.2  420.91
#Mann=11,-1,0
  4455.0    0.05       0  4727.5     0.1       0  4831.3    0.15       0
  4840.5    0.05       0  4857.5    0.07       0  4864.3    0.05       0
  4935.1     0.1       0  5145.5    0.08       0  5244.7     0.1       0
  5426.7    0.08       0  5624.0    0.05       0
Bank Sta=4759,5419.6
Exp/Cntr=0.3,0.1

Type RM Length L Ch R = 1,7946,499,499,499
BEGIN DESCRIPTION:
Mapping XS 61f78c62
END DESCRIPTION:
XS GIS Cut Line= 4
      2837828.65      7017944.64      2837623.79      7017521.04
      2837543.93      7017305.76      2837422.52      7016629.32
#Sta/Elev= 30
  4311.7  416.34  4322.4  416.44  4348.5  414.29  4363.0  414.04  4425.7  412.53
  4442.7  411.53  4448.3  412.09  4465.3  411.00  4470.9  411.50  4493.5  411.17
  4565.4  409.39  4582.8  408.81  4644.5  406.91  4747.5  405.73  4782.5  403.96
  4801.8  403.34  4877.1  401.28  4907.1  400.80  4961.8  399.21  4962.3  398.41
  4968.1  398.41  4968.6  399.21  5373.5  399.23  5411.6  401.18  5413.7  401.28
  5432.3  401.69  5486.0  406.33  5511.5  407.72  5657.3  415.81  5699.1  420.46
#Mann=12,-1,0
  4311.7    0.05       0  4348.5    0.08       0  4363.0    0.05       0
  4565.4    0.08       0  4582.8    0.05       0  4782.5    0.08       0
  4801.8     0.1       0  4907.1    0.05       0  4961.8   0.033       0
  4968.6    0.05       0  5411.6    0.16       0  5511.5    0.05       0
Bank Sta=4877.1,5413.7
Exp/Cntr=0.3,0.1

Type RM Length L Ch R = 1,7447,521,521,521
BEGIN DESCRIPTION:
Penson Spring Branch 13.0
END DESCRIPTION:
XS GIS Cut Line= 3
      2837975.00      7017924.95      2838025.00      7017175.00
      2838275.01      7016374.97
#Sta/Elev= 30
  4245.2  418.29  4275.2  417.49  4345.4  413.12  4565.9  402.87  4586.9  401.19
  4612.5  399.21  4613.0  398.41  4618.9  398.41  4619.4  399.21  5374.0  399.21
  5409.0  401.19  5445.8  403.31  5483.5  404.70  5548.4  408.68  5553.7  408.41
  5580.9  409.70  5586.1  409.54  5618.6  411.54  5645.9  414.54  5651.1  414.51
  5656.9  415.37  5677.8  416.31  5688.8  417.41  5698.8  421.42  5709.2  423.30
  5721.3  423.77  5748.5  423.71  5813.5  422.96  5818.7  427.95  5835.0  428.45
#Mann=3,-1,0
  4245.2    0.05       0  4612.5   0.033       0  4619.4    0.05       0
Bank Sta=4586.9,5409
Exp/Cntr=0.3,0.1

Type RM Length L Ch R = 1,6926,516,516,516
BEGIN DESCRIPTION:
Penson Spring Branch 12.0
END DESCRIPTION:
XS GIS Cut Line= 3
      2838725.01      7017625.03      2838525.00      7017025.00
      2838325.01      7016425.04
#Sta/Elev= 30
  4378.5  419.31  4389.1  419.07  4410.2  417.43  4420.7  417.03  4431.2  415.50
  4452.3  413.84  4462.9  412.43  4526.1  405.65  4547.2  404.39  4557.7  404.77
  4568.3  402.88  4584.8  401.86  4594.1  401.12  4617.5  399.21  4618.0  398.41
  4623.9  398.41  4624.4  399.21  5348.3  399.21  5373.2  401.12  5432.6  405.27
  5464.2  408.04  5495.9  411.59  5506.4  413.04  5538.0  416.15  5559.1  417.81
  5569.7  419.30  5590.7  421.40  5622.4  426.02  5632.9  427.82  5643.4  428.36
#Mann=4,-1,0
  4378.5    0.16       0  4584.8    0.05       0  4617.5   0.033       0
  4624.4    0.05       0
Bank Sta=4594.1,5373.2
Exp/Cntr=0.3,0.1

Type RM Length L Ch R = 1,6410,576,576,576
BEGIN DESCRIPTION:
Penson Spring Branch 11.0
END DESCRIPTION:
XS GIS Cut Line= 3
      2839375.03      7017275.03      2839025.00      7016875.00
      2838424.99      7016324.99
#Sta/Elev= 30
  4454.1  415.32  4475.5  414.35  4553.3  406.36  4581.8  404.60  4588.4  403.29
  4616.0  401.04  4635.3  399.21  4635.8  398.41  4641.7  398.41  4642.2  399.21
  5319.5  399.21  5360.9  399.21  5381.1  401.04  5424.4  403.65  5431.8  403.22
  5436.8  404.11  5466.9  406.65  5495.3  407.54  5516.3  409.81  5537.8  410.01
  5544.6  410.98  5552.0  410.20  5580.4  412.27  5587.2  413.79  5594.6  413.61
  5601.3  415.10  5615.5  416.36  5658.1  417.98  5771.5  427.35  5799.6  428.28
#Mann=5,-1,0
  4454.1    0.05       0  4635.3   0.033       0  4642.2    0.05       0
  5319.5    0.16       0  5436.8    0.05       0
Bank Sta=4616,5381.1
Exp/Cntr=0.3,0.1

Type RM Length L Ch R = 1,5834,502,502,502
BEGIN DESCRIPTION:
Penson Spring Branch 10.0
END DESCRIPTION:
XS GIS Cut Line= 3
      2839425.00      7017275.00      2839575.00      7016775.00
      2839125.00      7015974.99
#Sta/Elev= 30
  4484.3  415.18  4557.4  412.26  4599.1  408.93  4610.5  407.56  4661.8  404.25
  4684.0  400.94  4706.1  399.21  4706.6  398.41  4712.6  398.41  4713.1  399.21
  5570.7  399.21  5602.6  401.56  5608.5  400.94  5624.3  403.02  5630.0  402.43
  5646.0  404.64  5673.4  405.75  5689.3  407.32  5754.3  411.34  5770.3  412.85
  5791.9  413.78  5807.9  415.58  5856.9  419.21  5872.9  421.16  5888.8  422.03
  5894.6  421.86  5910.5  424.19  5916.2  424.47  5921.3  426.36  5924.2  426.36
#Mann=3,-1,0
  4484.3    0.05       0  4706.1   0.033       0  4713.1    0.05       0
Bank Sta=4684,5608.5
Exp/Cntr=0.3,0.1

Type RM Length L Ch R = 1,5332,579,579,579
BEGIN DESCRIPTION:
Penson Spring Branch 9.0
END DESCRIPTION:
XS GIS Cut Line= 3
      2839624.97      7017525.04      2840068.23      7016878.68
      2839870.54      7016119.13
#Sta/Elev= 30
  4209.7  416.45  4274.0  413.95  4303.8  412.00  4324.8  411.88  4331.0  410.80
  4354.6  410.11  4367.4  406.11  4381.6  404.88  4390.5  405.08  4396.5  406.66
  4403.8  407.49  4411.5  406.48  4432.4  405.66  4483.2  401.87  4504.2  400.87
  4515.5  399.21  4516.1  398.41  4522.1  398.41  4522.6  399.21  5513.9  399.21
  5524.2  399.35  5541.4  400.87  5546.2  401.58  5565.6  402.36  5586.7  405.13
  5616.9  406.36  5627.6  407.57  5657.4  408.44  5743.6  414.52  5778.3  415.18
#Mann=3,-1,0
  4209.7    0.05       0  4515.5   0.033       0  4522.6    0.05       0
Bank Sta=4504.2,5541.4
Exp/Cntr=0.3,0.1

Type RM Length L Ch R = 1,4753,522,522,522
BEGIN DESCRIPTION:
Penson Spring Branch 8.0
END DESCRIPTION:
XS GIS Cut Line= 3
      2840175.00      7017825.00      2840625.00      7017025.00
      2840925.01      7016224.98
#Sta/Elev= 30
  4085.2  416.48  4195.8  414.21  4336.6  406.72  4371.6  404.14  4379.4  403.63
  4385.1  401.95  4401.0  402.65  4406.8  401.85  4417.0  402.00  4422.7  400.93
  4438.8  400.76  4444.4  399.53  4462.1  399.21  4462.8  398.41  4469.4  398.41
  4470.0  399.21  5360.0  399.23  5378.2  400.76  5383.3  400.82  5390.2  400.91
  5398.2  404.35  5500.6  410.59  5586.0  410.86  5616.3  411.46  5641.2  413.07
  5665.5  413.27  5718.6  415.76  5787.2  417.51  5849.8  421.71  5857.5  422.06
#Mann=8,-1,0
  4085.2    0.05       0  4336.6    0.16       0  4371.6    0.05       0
  4462.1   0.033       0  4470.0    0.05       0  5383.3    0.16       0
  5665.5    0.05       0  5849.8    0.08       0
Bank Sta=4438.8,5378.2
Exp/Cntr=0.3,0.1

Type RM Length L Ch R = 1,4231,536,536,536
BEGIN DESCRIPTION:
Penson Spring Branch 7.0
END DESCRIPTION:
XS GIS Cut Line= 3
      2840574.98      7017975.03      2841125.00      7017175.00
      2841175.00      7016425.03
#Sta/Elev= 30
  4032.4  415.47  4039.9  415.46  4045.6  416.24  4060.8  415.70  4068.8  414.49
  4081.8  413.27  4153.8  409.33  4177.2  408.61  4204.3  406.36  4226.6  405.85
  4248.9  404.67  4255.0  404.85  4269.9  404.39  4284.8  403.07  4299.4  402.71
  4326.7  401.19  4345.3  400.62  4373.5  399.21  4374.2  398.41  4380.8  398.41
  4381.4  399.21  4396.6  399.21  5514.4  399.21  5554.7  400.62  5564.5  404.65
  5593.9  405.36  5624.6  407.30  5684.8  412.15  5714.8  414.04  5754.9  414.97
#Mann=6,-1,0
  4032.4    0.05       0  4045.6    0.16       0  4373.5   0.033       0
  4381.4    0.16       0  4396.6    0.05       0  5593.9    0.16       0
Bank Sta=4345.3,5554.7
Exp/Cntr=0.3,0.1

Type RM Length L Ch R = 1,3695,544,544,544
BEGIN DESCRIPTION:
Penson Spring Branch 6.0
END DESCRIPTION:
XS GIS Cut Line= 3
      2840475.03      7018174.98      2841625.00      7017375.00
      2842424.98      7016575.02
#Sta/Elev= 30
  3607.2  419.99  3721.9  419.10  3729.0  418.38  3736.8  418.97  3889.0  414.76
  3966.3  411.78  3996.0  412.23  4002.1  411.41  4017.0  412.02  4037.9  411.16
  4067.6  412.16  4073.7  411.38  4088.5  411.85  4139.2  410.56  4246.5  406.86
  4267.4  405.48  4275.4  403.49  4282.3  403.37  4289.3  401.41  4305.0  400.52
  4321.9  399.21  4322.6  398.41  4329.2  398.41  4329.8  399.21  5884.9  399.21
  5918.2  400.32  5928.0  400.52  5941.4  404.46  6082.9  413.34  6139.4  415.43
#Mann=7,-1,0
  3607.2    0.16       0  3736.8    0.12       0  3889.0    0.16       0
  4275.4    0.05       0  4321.9   0.033       0  4329.8    0.05       0
  5918.2    0.16       0
Bank Sta=4305,5928
Exp/Cntr=0.3,0.1
