HEC-RAS study SCHOOLEY CREEK.prj: SCHOOLEY CREEK Base Level Engineering

--- SCHOOLEY CREEK.g01 (geometry) --- (continued)

Type RM Length L Ch R = 1,61164,276,276,276
BEGIN DESCRIPTION:
Mapping XS 7ac767ed
END DESCRIPTION:
XS GIS Cut Line= 3
      2794998.06      7080708.82      2794638.67      7080656.73
      2794081.42      7080646.32
#Sta/Elev= 30
  4651.6  519.43  4716.7  519.06  4796.2  516.29  4826.5  517.05  4857.2  516.67
  4877.0  517.02  4908.7  516.21  4917.3  515.49  4923.6  513.95  4927.5  511.90
  4957.8  511.52  4978.0  512.04  4987.5  510.87  4992.6  509.16  4994.0  503.48
  4994.7  502.68  5001.7  502.68  5002.5  503.48  5008.4  509.96  5014.1  512.38
  5068.4  512.38  5138.4  513.14  5148.4  509.88  5158.4  510.93  5168.4  513.19
  5228.5  513.31  5292.6  512.73  5370.9  513.95  5468.5  515.69  5572.1  518.63
#Mann=5,-1,0
  4651.6    0.05       0  4908.7    0.12       0  4994.0    0.07       0
  5002.5    0.12       0  5292.6    0.16       0
Bank Sta=4923.6,5370.9
Exp/Cntr=0.3,0.1

Type RM Length L Ch R = 1,60888,413,413,413
BEGIN DESCRIPTION:
Mapping XS 73adc2a7
END DESCRIPTION:
XS GIS Cut Line= 3
      2795055.38      7080437.98      2794617.83      7080417.15
      2794065.74      7080281.73
#Sta/Elev= 30
  4546.1  520.01  4666.6  518.17  4696.6  518.45  4717.8  517.47  4756.7  517.81
  4827.7  514.99  4856.2  513.56  4896.9  511.98  4916.9  512.11  4928.1  510.73
  4988.2  510.93  5003.4  503.02  5004.1  502.22  5011.1  502.22  5011.9  503.02
  5013.5  509.72  5028.2  511.47  5061.6  511.66  5079.7  512.19  5138.2  510.94
  5199.6  511.68  5221.4  511.73  5226.5  509.36  5234.2  508.81  5268.1  512.02
  5368.0  512.55  5383.7  513.56  5398.9  516.30  5409.2  517.00  5552.6  519.62
#Mann=6,-1,0
  4546.1    0.05       0  4827.7    0.12       0  5003.4    0.07       0
  5011.9    0.12       0  5061.6    0.16       0  5199.6    0.05       0
Bank Sta=4856.2,5383.7
Exp/Cntr=0.3,0.1

Type RM Length L Ch R = 1,60475,322,322,322
BEGIN DESCRIPTION:
Mapping XS c6ccfbf8
END DESCRIPTION:
XS GIS Cut Line= 3
      2795102.23      7080339.03      2794607.42      7080089.02
      2794164.76      7080047.36
#Sta/Elev= 30
  4458.4  520.13  4475.3  519.05  4533.7  519.40  4570.0  518.46  4586.7  519.31
  4623.4  519.49  4735.4  515.95  4756.6  511.69  4765.1  510.53  4793.3  510.34
  4854.2  509.51  4898.8  510.23  4914.7  508.14  4921.1  510.49  4926.7  510.82
  4981.9  510.64  4988.0  505.01  4989.2  502.87  4990.0  502.07  4997.1  502.07
  4997.9  502.87  5004.3  504.05  5010.3  510.88  5012.8  511.29  5128.3  511.01
  5175.9  510.54  5210.9  511.69  5406.9  518.35  5430.6  517.87  5457.4  518.82
#Mann=5,-1,0
  4458.4    0.05       0  4793.3    0.12       0  4989.2    0.07       0
  4997.9    0.12       0  5128.3    0.05       0
Bank Sta=4756.6,5210.9
Exp/Cntr=0.3,0.1

Type RM Length L Ch R = 1,60153,383,383,383
BEGIN DESCRIPTION:
Mapping XS 3781ebbd
END DESCRIPTION:
XS GIS Cut Line= 3
      2795216.77      7080109.84      2794737.62      7079828.61
      2794253.20      7079698.39
#Sta/Elev= 30
  4431.4  519.27  4503.0  518.99  4589.6  516.55  4648.2  513.47  4756.0  511.58
  4882.7  509.41  4932.0  510.90  4978.4  510.14  4981.3  500.41  4982.1  499.61
  4989.2  499.61  4990.0  500.41  5000.1  501.11  5010.4  507.45  5017.9  510.13
  5041.5  510.60  5057.8  509.26  5063.0  509.95  5072.5  507.68  5092.6  509.06
  5145.0  506.48  5155.4  508.45  5165.7  509.03  5238.2  509.87  5281.1  511.58
  5327.3  513.30  5367.2  513.05  5407.2  515.99  5455.7  517.58  5488.6  517.65
#Mann=3,-1,0
  4431.4    0.05       0  4981.3    0.03       0  4990.0    0.05       0
Bank Sta=4756,5281.1
Exp/Cntr=0.3,0.1

Type RM Length L Ch R = 1,59770,525,525,525
BEGIN DESCRIPTION:
Mapping XS 0e0d6a56
END DESCRIPTION:
XS GIS Cut Line= 3
      2795331.39      7080063.00      2794945.96      7079542.15
      2794608.68      7079355.35
#Sta/Elev= 30
  4357.8  518.46  4554.4  516.04  4604.1  513.54  4625.9  513.70  4684.3  511.23
  4789.1  509.61  4847.2  509.87  4876.4  508.79  4976.6  508.43  4982.8  504.64
  4993.1  500.60  4993.9  499.80  5001.1  499.80  5001.8  500.60  5002.4  505.82
  5008.0  505.82  5011.4  507.87  5018.3  508.34  5054.9  509.04  5086.9  508.32
  5136.2  508.90  5189.7  507.57  5214.5  510.70  5218.2  511.23  5224.0  512.73
  5246.9  516.03  5261.0  516.90  5292.6  517.45  5314.8  518.78  5391.3  518.53
#Mann=5,-1,0
  4357.8    0.05       0  4789.1    0.16       0  4993.1    0.07       0
  5001.8    0.16       0  5214.5    0.05       0
Bank Sta=4684.3,5218.2
Exp/Cntr=0.3,0.1

Type RM Length L Ch R = 1,59245,473,473,473
BEGIN DESCRIPTION:
Mapping XS 4c072483
END DESCRIPTION:
XS GIS Cut Line= 3
      2795607.43      7079979.69      2795409.50      7079406.73
      2795045.50      7079089.53
#Sta/Elev= 30
  4404.6  518.66  4504.8  516.90  4551.1  514.54  4621.2  513.37  4663.5  510.84
  4708.9  509.92  4726.6  509.48  4908.6  507.79  4951.2  506.48  4959.7  507.47
  4977.1  507.30  4982.4  504.93  4987.0  497.53  4987.9  496.73  4995.1  496.73
  4995.9  497.53  5002.0  503.28  5008.3  507.81  5010.8  508.58  5029.8  509.16
  5036.4  508.29  5077.0  507.36  5107.7  506.73  5128.5  507.50  5205.7  507.70
  5283.2  509.92  5327.0  511.06  5355.4  513.67  5398.2  515.38  5493.6  517.24
#Mann=7,-1,0
  4404.6    0.05       0  4726.6    0.16       0  4908.6    0.12       0
  4987.0    0.07       0  4995.9    0.12       0  5077.0    0.16       0
  5205.7    0.05       0
Bank Sta=4708.9,5283.2
Exp/Cntr=0.3,0.1

Type RM Length L Ch R = 1,58772,606,606,606
BEGIN DESCRIPTION:
Mapping XS cedcf879
END DESCRIPTION:
XS GIS Cut Line= 3
      2796024.11      7079130.69      2795633.46      7079073.40
      2795118.91      7079021.42
#Sta/Elev= 30
  4606.0  514.91  4675.2  513.39  4716.1  513.39  4764.9  513.93  4787.0  513.76
  4864.9  509.24  4870.7  509.06  4908.3  507.74  4928.5  506.10  4959.6  506.18
  4979.1  507.02  4989.2  500.10  4992.9  498.29  4993.8  497.49  5001.2  497.49
  5002.1  498.29  5009.3  504.68  5019.4  506.39  5079.7  506.65  5119.9  504.52
  5134.6  506.57  5140.0  506.51  5190.2  504.19  5200.3  507.16  5202.8  507.12
  5260.6  506.98  5348.3  509.24  5434.6  512.32  5481.7  517.02  5518.0  516.89
#Mann=7,-1,0
  4606.0    0.16       0  4716.1    0.12       0  4764.9    0.16       0
  4870.7    0.12       0  4992.9    0.07       0  5002.1    0.12       0
  5202.8    0.05       0
Bank Sta=4864.9,5348.3
Exp/Cntr=0.3,0.1

Type RM Length L Ch R = 1,58166,435,435,435
BEGIN DESCRIPTION:
Mapping XS eff255d8
END DESCRIPTION:
XS GIS Cut Line= 3
      2796065.80      7078672.35      2795643.87      7078714.02
      2795133.50      7078901.51
#Sta/Elev= 30
  4555.3  512.76  4596.3  512.96  4632.3  512.32  4696.8  513.02  4738.4  512.83
  4757.1  513.29  4819.1  510.92  4856.7  507.47  4867.6  506.11  4877.7  505.47
  4940.7  506.74  4968.1  506.14  4976.2  504.64  4981.3  504.64  4988.7  501.67
  4995.3  496.62  4996.1  496.35  4996.9  495.55  5004.4  495.55  5005.3  496.35
  5007.0  498.52  5010.0  502.35  5025.8  505.12  5228.4  506.70  5295.9  507.47
  5370.3  508.62  5425.5  510.15  5486.9  513.65  5492.2  513.45  5523.0  516.40
#Mann=6,-1,0
  4555.3    0.16       0  4819.1    0.12       0  4996.1    0.07       0
  5005.3    0.12       0  5007.0    0.16       0  5228.4    0.05       0
Bank Sta=4856.7,5295.9
Exp/Cntr=0.3,0.1

Type RM Length L Ch R = 1,57731,869,869,869
BEGIN DESCRIPTION:
Mapping XS dbd7e08e
END DESCRIPTION:
XS GIS Cut Line= 3
      2796076.19      7078615.08      2795633.46      7078432.77
      2795044.95      7078182.79
#Sta/Elev= 30
  4498.5  511.89  4644.5  511.14  4692.4  512.41  4745.7  511.34  4774.6  509.21
  4808.8  506.74  4867.5  505.45  4889.1  504.04  4982.7  504.07  4992.7  496.35
  4993.6  495.55  5001.1  495.55  5001.9  496.35  5019.1  504.79  5149.5  504.84
  5159.2  502.07  5164.6  504.55  5171.2  500.65  5182.1  501.76  5188.2  504.17
  5193.7  503.39  5203.8  505.35  5258.1  503.80  5311.0  503.83  5420.7  506.68
  5425.3  506.74  5475.6  507.53  5493.8  509.08  5592.2  512.27  5616.7  512.90
#Mann=7,-1,0
  4498.5    0.16       0  4774.6    0.12       0  4992.7    0.07       0
  5001.9    0.12       0  5311.0    0.05       0  5420.7    0.12       0
  5592.2    0.16       0
Bank Sta=4808.8,5425.3
Exp/Cntr=0.3,0.1

Type RM Length L Ch R = 1,56862,529,529,529
BEGIN DESCRIPTION:
Mapping XS db7d5bde
END DESCRIPTION:
XS GIS Cut Line= 3
      2796383.45      7078427.56      2795810.54      7077948.40
      2795368.90      7077465.20
#Sta/Elev= 30
  4225.1  512.68  4553.9  507.20  4588.1  506.95  4601.5  510.20  4615.8  505.78
  4658.8  509.02  4673.1  505.57  4689.8  507.72  4736.9  505.04  4751.2  508.71
  4761.7  504.86  4815.4  503.91  4956.8  503.05  4978.1  501.71  4985.5  496.19
  5001.6  493.99  5002.6  493.19  5011.2  493.99  5013.9  498.93  5020.6  503.38
  5028.0  504.11  5077.4  502.09  5119.9  504.22  5134.1  499.72  5240.2  503.95
  5396.6  504.86  5434.1  508.10  5466.5  512.74  5530.6  508.90  5626.6  511.65
#Mann=7,-1,0
  4225.1    0.05       0  4553.9    0.16       0  4689.8    0.12       0
  4815.4    0.16       0  5001.6    0.07       0  5011.2    0.16       0
  5434.1    0.05       0
Bank Sta=4761.7,5396.6
Exp/Cntr=0.3,0.1

Type RM Length L Ch R = 1,56333,514,514,514
BEGIN DESCRIPTION:
SCHOOLEY CREEK 53.0
END DESCRIPTION:
XS GIS Cut Line= 3
      2796525.01      7078225.02      2796275.00      7077775.00
      2795725.01      7077275.01
#Sta/Elev= 30
  4494.2  511.19  4545.7  508.96  4561.7  509.88  4567.4  508.37  4583.5  509.12
  4589.2  507.36  4605.2  509.09  4610.9  507.60  4626.9  508.67  4729.2  505.82
  4848.5  503.54  4982.1  501.21  4986.1  500.80  4996.2  493.38  4997.1  492.58
  5005.9  493.38  5006.1  497.68  5012.4  497.68  5016.1  501.31  5018.4  501.48
  5093.8  501.40  5157.7  503.01  5171.5  502.87  5180.9  500.00  5214.1  500.02
  5235.7  501.60  5384.2  501.20  5466.3  501.90  5496.6  503.54  5752.3  512.71
#Mann=9,-1,0
  4494.2    0.05       0  4729.2    0.16       0  4982.1    0.12       0
  4996.2    0.07       0  5005.9    0.12       0  5018.4    0.16       0
  5180.9    0.12       0  5384.2    0.16       0  5466.3    0.05       0
Bank Sta=4848.5,5496.6
Exp/Cntr=0.3,0.1

Type RM Length L Ch R = 1,55819,544,544,544
BEGIN DESCRIPTION:
SCHOOLEY CREEK 52.0
END DESCRIPTION:
XS GIS Cut Line= 3
      2796725.00      7078124.96      2796675.00      7077475.00
      2796275.00      7076874.99
#Sta/Elev= 30
  4345.0  511.75  4386.5  510.46  4495.5  509.04  4525.5  509.84  4593.8  509.59
  4635.8  509.50  4836.3  502.36  4885.8  500.69  4926.7  499.98  4976.8  500.81
  4994.4  494.51  4996.9  494.51  4999.5  493.01  5000.5  492.21  5008.3  492.21
  5009.2  493.01  5010.4  499.08  5019.4  500.63  5076.5  499.88  5133.6  500.83
  5141.1  499.96  5154.6  496.24  5177.2  498.83  5241.8  500.54  5307.9  500.19
  5386.4  502.36  5416.6  503.65  5452.1  505.39  5566.3  507.15  5718.0  510.87
#Mann=8,-1,0
  4345.0    0.16       0  4386.5    0.05       0  4495.5    0.12       0
  4593.8    0.16       0  4885.8    0.12       0  4999.5    0.07       0
  5009.2    0.12       0  5416.6    0.16       0
Bank Sta=4836.3,5386.4
Exp/Cntr=0.3,0.1

Type RM Length L Ch R = 1,55275,445,445,445
BEGIN DESCRIPTION:
SCHOOLEY CREEK 51.0
END DESCRIPTION:
XS GIS Cut Line= 3
      2796925.00      7078225.05      2797025.00      7077125.00
      2796424.99      7076725.00
#Sta/Elev= 30
  3875.5  511.53  3960.8  510.50  4135.5  508.22  4335.8  504.93  4468.0  505.27
  4634.6  501.11  4799.3  498.45  4950.0  499.62  4970.0  498.63  4977.6  494.23
  4983.1  494.23  4987.6  496.90  4993.6  491.30  4997.6  490.96  4998.6  490.16
  5007.6  490.96  5008.6  495.96  5044.7  499.23  5052.2  498.73  5059.7  495.18
  5065.7  497.42  5074.7  496.01  5116.8  499.86  5288.0  500.44  5297.1  501.11
  5439.9  505.68  5672.6  511.64  5678.7  509.44  5693.7  508.54  5701.2  510.47
#Mann=8,-1,0
  3875.5    0.16       0  3960.8    0.05       0  4135.5    0.16       0
  4335.8    0.12       0  4997.6    0.07       0  5007.6    0.12       0
  5288.0    0.16       0  5439.9    0.05       0
Bank Sta=4634.6,5297.1
Exp/Cntr=0.3,0.1

Type RM Length L Ch R = 1,54830,1471,1471,1471
BEGIN DESCRIPTION:
SCHOOLEY CREEK 50.0
END DESCRIPTION:
XS GIS Cut Line= 3
      2797289.71      7077573.35      2797258.46      7076911.94
      2796915.46      7076298.70
#Sta/Elev= 30
  4298.5  506.48  4372.6  504.73  4397.0  504.39  4437.0  505.77  4497.1  504.15
  4547.1  505.85  4577.2  505.03  4607.2  506.04  4637.2  504.62  4707.3  503.81
  4735.0  501.86  4785.8  500.34  4807.4  499.85  4827.4  497.41  4837.5  497.32
  4907.5  499.08  4968.6  499.02  4981.9  495.96  4986.5  488.76  4987.5  487.96
  4995.5  487.96  4996.5  488.76  5003.6  494.57  5013.8  498.41  5136.0  498.06
  5188.0  497.27  5269.2  498.28  5415.2  500.04  5444.6  500.34  5663.3  507.09
#Mann=9,-1,0
  4298.5    0.05       0  4372.6    0.16       0  4735.0    0.12       0
  4986.5    0.07       0  4996.5    0.12       0  5136.0    0.16       0
  5188.0    0.05       0  5269.2    0.16       0  5415.2    0.05       0
Bank Sta=4785.8,5444.6
Exp/Cntr=0.3,0.1

Type RM Length L Ch R = 1,53359,740,740,740
BEGIN DESCRIPTION:
SCHOOLEY CREEK 49.0
END DESCRIPTION:
XS GIS Cut Line= 3
      2798025.02      7076925.02      2797725.00      7076575.00
      2797074.98      7076124.99
#Sta/Elev= 30
  4552.8  506.40  4637.9  505.29  4645.0  504.02  4744.4  500.75  4765.7  498.30
  4793.7  495.82  4808.0  496.62  4815.7  498.39  4822.3  497.80  4836.6  500.90
  4867.5  500.88  4893.6  500.16  4935.3  496.34  4985.8  495.71  4992.4  493.15
  4995.1  486.96  4996.1  486.16  5005.1  486.96  5006.7  486.99  5010.5  493.81
  5016.8  493.81  5021.2  496.75  5162.0  496.19  5221.2  495.17  5442.8  497.15
  5522.5  498.30  5626.7  501.17  5631.9  501.37  5689.5  504.19  5804.4  506.59
#Mann=8,-1,0
  4552.8    0.05       0  4867.5    0.12       0  4995.1    0.07       0
  5005.1    0.12       0  5162.0    0.05       0  5442.8    0.12       0
  5626.7    0.16       0  5631.9    0.05       0
Bank Sta=4765.7,5522.5
Exp/Cntr=0.3,0.1

Type RM Length L Ch R = 1,52619,844,844,844
BEGIN DESCRIPTION:
Mapping XS 1b70d985
END DESCRIPTION:
XS GIS Cut Line= 3
      2798211.57      7076656.71      2797972.00      7076281.73
      2797435.50      7075964.00
#Sta/Elev= 30
  4569.8  506.66  4741.9  504.56  4929.1  497.39  4935.3  497.33  4975.3  495.62
  4987.2  485.74  4996.5  486.30  5002.4  492.16  5009.9  494.04  5054.7  494.90
  5076.1  493.82  5081.9  487.91  5091.8  492.62  5092.6  485.23  5093.5  484.43
  5101.6  484.43  5102.6  485.23  5104.3  492.77  5113.2  494.65  5119.0  493.29
  5127.5  495.38  5171.7  494.01  5296.3  494.37  5332.9  493.57  5460.2  497.39
  5492.0  498.02  5541.3  499.60  5580.8  501.15  5586.9  502.27  5638.3  503.45
#Mann=8,-1,0
  4569.8    0.05       0  4935.3    0.12       0  5092.6    0.07       0
  5102.6    0.12       0  5296.3    0.05       0  5332.9    0.12       0
  5492.0    0.16       0  5541.3    0.05       0
Bank Sta=4929.1,5460.2
Exp/Cntr=0.3,0.1

Type RM Length L Ch R = 1,51775,506,506,506
BEGIN DESCRIPTION:
SCHOOLEY CREEK 47.0
END DESCRIPTION:
XS GIS Cut Line= 3
      2798775.01      7076375.01      2798375.00      7076125.00
      2797674.99      7075674.99
#Sta/Elev= 30
  4528.5  506.64  4709.5  504.84  4954.1  498.60  4971.3  499.34  4981.5  495.40
  4986.7  492.80  4987.5  486.67  4988.5  485.87  4997.6  486.67  5007.8  487.60
  5013.8  490.67  5028.9  493.68  5035.9  493.90  5131.0  494.33  5180.2  493.05
  5202.3  494.22  5261.8  493.72  5304.4  494.99  5377.0  493.50  5413.3  494.48
  5428.2  491.47  5434.5  493.86  5440.4  494.39  5528.2  492.88  5579.8  493.50
  5619.5  495.40  5640.7  496.17  5785.6  501.77  5822.7  503.14  5832.4  503.19
#Mann=7,-1,0
  4528.5    0.05       0  4954.1    0.12       0  4987.5    0.07       0
  4997.6    0.12       0  5640.7    0.16       0  5785.6    0.05       0
  5822.7    0.16       0
Bank Sta=4981.5,5619.5
Exp/Cntr=0.3,0.1

Type RM Length L Ch R = 1,51269,599,599,599
BEGIN DESCRIPTION:
Mapping XS 2390259d
END DESCRIPTION:
XS GIS Cut Line= 3
      2798904.30      7075995.28      2798701.17      7075880.69
      2797720.05      7075589.99
#Sta/Elev= 30
  4782.5  504.29  4957.9  501.69  4965.4  500.73  4973.8  498.16  4980.6  494.16
  4988.4  488.34  4990.4  484.95  4991.4  484.15  4999.5  484.15  5000.5  484.95
  5010.7  491.76  5033.7  492.33  5265.9  493.16  5272.5  492.81  5282.9  488.45
  5293.3  486.65  5304.4  487.67  5314.2  487.13  5324.6  488.76  5345.5  488.87
  5370.9  493.29  5376.8  493.46  5491.5  492.35  5620.3  492.75  5652.5  491.45
  5685.7  493.10  5754.3  494.16  5929.1  498.05  6031.7  502.21  6039.0  502.31
#Mann=7,-1,0
  4782.5    0.05       0  4990.4    0.03       0  5000.5    0.05       0
  5033.7    0.12       0  5620.3    0.16       0  5929.1    0.05       0
  6031.7    0.16       0
Bank Sta=4980.6,5754.3
Exp/Cntr=0.3,0.1

Type RM Length L Ch R = 1,50670,526,526,526
BEGIN DESCRIPTION:
Mapping XS 21576f1e
END DESCRIPTION:
XS GIS Cut Line= 3
      2798940.74      7075812.97      2798544.92      7075432.77
      2798129.64      7074960.40
#Sta/Elev= 30
  4423.2  503.48  4546.0  499.87  4638.1  499.71  4687.3  493.54  4706.9  492.96
  4885.6  490.72  4972.0  491.68  4977.6  491.48  4984.3  488.01  4991.8  489.57
  4998.5  482.93  5001.0  482.86  5002.0  482.06  5011.1  482.86  5012.7  485.87
  5020.3  486.18  5027.0  491.05  5034.5  484.28  5041.2  485.11  5048.8  491.18
  5055.4  488.76  5062.3  491.81  5161.7  489.29  5175.9  483.93  5182.6  484.80
  5190.1  490.13  5211.0  492.57  5394.6  493.54  5425.8  495.86  5601.0  500.44
#Mann=5,-1,0
  4423.2    0.05       0  4706.9    0.12       0  5001.0    0.07       0
  5011.1    0.12       0  5425.8    0.16       0
Bank Sta=4687.3,5394.6
Exp/Cntr=0.3,0.1

Type RM Length L Ch R = 1,50144,1152,1152,1152
BEGIN DESCRIPTION:
Mapping XS 379c79c3
END DESCRIPTION:
XS GIS Cut Line= 3
      2799133.45      7075667.13      2798930.33      7075354.65
      2798221.97      7074901.50
#Sta/Elev= 30
  4606.5  503.41  4780.0  500.06  4823.7  497.86  4873.4  492.27  4888.7  490.72
  4911.9  490.59  4954.9  490.89  4961.2  487.48  4967.1  490.19  4976.0  487.51
  4983.7  489.35  4997.4  483.17  5004.9  483.77  5010.8  488.74  5020.1  490.47
  5104.7  489.87  5222.9  492.10  5301.7  491.98  5353.3  489.96  5453.1  489.64
  5460.4  487.36  5463.3  482.98  5464.2  482.18  5473.4  482.98  5474.2  488.32
  5483.5  490.22  5504.7  491.87  5619.8  492.27  5649.1  492.89  5820.1  498.99
#Mann=5,-1,0
  4606.5    0.05       0  4911.9    0.12       0  5463.3    0.07       0
  5473.4    0.12       0  5649.1    0.16       0
Bank Sta=4873.4,5619.8
Exp/Cntr=0.3,0.1

Type RM Length L Ch R = 1,48992,506,506,506
BEGIN DESCRIPTION:
SCHOOLEY CREEK 43.0
END DESCRIPTION:
XS GIS Cut Line= 3
      2799325.00      7075225.00      2798825.00      7074875.00
      2798325.02      7074825.00
#Sta/Elev= 30
  4398.6  500.31  4614.4  492.04  4705.0  490.49  4787.0  487.91  4873.3  489.72
  4950.9  488.67  4972.3  489.55  4980.6  488.28  4986.7  488.70  5000.7  479.68
  5001.6  478.88  5010.2  478.88  5011.1  479.68  5019.0  485.04  5029.0  488.61
  5032.0  488.77  5079.3  488.80  5089.3  487.59  5099.4  482.20  5109.4  481.56
  5119.5  484.64  5139.6  484.55  5157.2  490.00  5188.3  490.49  5223.5  492.04
  5275.3  490.86  5310.4  490.57  5368.3  492.12  5390.8  491.87  5511.4  496.37
#Mann=7,-1,0
  4398.6    0.05       0  5000.7    0.03       0  5011.1    0.05       0
  5032.0    0.12       0  5223.5    0.16       0  5275.3    0.12       0
  5368.3    0.16       0
Bank Sta=4705,5188.3
Exp/Cntr=0.3,0.1

Type RM Length L Ch R = 1,48486,792,792,792
BEGIN DESCRIPTION:
Mapping XS 95c5c224
END DESCRIPTION:
XS GIS Cut Line= 3
      2799414.73      7074906.75      2799086.58      7074609.86
      2798513.64      7074255.67
#Sta/Elev= 30
  4571.5  497.26  4657.4  496.16  4826.7  490.13  4883.9  487.73  4969.0  488.07
  4975.8  486.00  4983.2  478.96  4984.8  478.53  4985.7  477.73  4994.3  477.73
  4995.2  478.53  4997.4  481.73  5004.2  485.72  5013.9  488.73  5054.4  488.19
  5106.4  490.10  5228.2  487.86  5251.0  486.70  5264.8  488.10  5298.9  488.09
  5353.5  489.15  5374.8  490.37  5397.3  490.13  5398.0  490.17  5414.7  490.61
  5469.3  490.92  5529.5  492.59  5599.3  494.73  5643.1  496.33  5687.6  496.37
#Mann=8,-1,0
  4571.5    0.05       0  4984.8    0.07       0  4995.2    0.05       0
  5298.9    0.16       0  5398.0    0.12       0  5414.7    0.16       0
  5529.5    0.12       0  5599.3    0.05       0
Bank Sta=4826.7,5397.3
Exp/Cntr=0.3,0.1

Type RM Length L Ch R = 1,47694,660,660,660
BEGIN DESCRIPTION:
Mapping XS c45b1784
END DESCRIPTION:
XS GIS Cut Line= 3
      2799982.39      7074792.14      2799649.08      7074609.86
      2798695.93      7074000.47
#Sta/Elev= 30
  4621.9  498.61  4772.5  494.45  4854.1  489.95  4859.8  491.27  4875.6  489.09
  4881.6  490.80  4892.0  489.42  4897.7  490.13  4957.5  481.98  4961.7  485.66
  4963.2  486.98  4972.3  480.39  4974.1  477.33  4975.0  476.53  4984.6  477.33
  5001.1  480.94  5007.2  479.85  5016.3  485.12  5022.3  481.10  5030.4  486.43
  5037.5  487.40  5219.3  488.27  5303.9  487.21  5485.8  489.32  5667.6  489.44
  5725.1  486.48  5820.4  487.15  5914.8  489.09  6088.1  494.41  6133.1  495.48
#Mann=6,-1,0
  4621.9    0.05       0  4961.7    0.12       0  4974.1    0.07       0
  4984.6    0.12       0  5820.4    0.16       0  6088.1    0.05       0
Bank Sta=4875.6,5914.8
Exp/Cntr=0.3,0.1

Type RM Length L Ch R = 1,47034,539,539,539
BEGIN DESCRIPTION:
Mapping XS b1785774
END DESCRIPTION:
XS GIS Cut Line= 3
      2800216.84      7074307.79      2799602.21      7074141.11
      2798765.53      7073969.61
#Sta/Elev= 30
  4319.5  494.93  4582.1  491.66  4697.6  488.37  4746.2  487.23  4810.6  489.36
  4845.3  486.13  4913.9  485.74  4936.4  485.37  4973.9  486.48  4984.1  482.75
  4989.1  475.82  4990.0  475.02  4999.6  475.82  5010.6  482.27  5015.7  479.82
  5024.9  482.83  5055.6  486.52  5061.1  486.29  5076.0  480.70  5086.2  480.89
  5116.8  486.37  5207.2  487.94  5290.3  488.04  5408.9  485.50  5504.6  487.66
  5545.1  486.94  5617.1  488.37  5643.3  489.06  5699.6  490.31  5810.4  493.77
#Mann=8,-1,0
  4319.5    0.05       0  4913.9    0.07       0  4936.4    0.12       0
  4989.1    0.07       0  4999.6    0.12       0  5545.1    0.16       0
  5643.3    0.12       0  5699.6    0.16       0
Bank Sta=4697.6,5617.1
Exp/Cntr=0.3,0.1

Type RM Length L Ch R = 1,46495,569,569,569
BEGIN DESCRIPTION:
XS2972A
END DESCRIPTION:
XS GIS Cut Line= 3
      2800018.88      7074172.36      2799591.79      7073823.40
      2798753.26      7073693.19
#Sta/Elev= 30
  4373.6  493.49  4502.5  489.42  4620.7  487.93  4715.0  484.94  4822.0  484.24
  4850.2  485.20  4925.1  485.73  4932.0  487.22  4982.6  485.15  4992.7  479.55
  4997.6  474.49  4998.5  473.69  5008.1  474.49  5010.2  481.03  5023.1  485.50
  5073.1  485.10  5078.2  483.17  5093.9  484.98  5114.2  482.69  5124.3  483.39
  5134.4  481.16  5141.1  483.94  5185.0  487.26  5227.7  486.47  5255.8  486.54
  5286.2  488.23  5366.3  487.93  5593.5  489.87  5615.4  490.02  5773.7  491.79
#Mann=7,-1,0
  4373.6    0.05       0  4850.2    0.12       0  4997.6    0.07       0
  5008.1    0.12       0  5227.7    0.16       0  5593.5    0.12       0
  5615.4    0.16       0
Bank Sta=4620.7,5366.3
Exp/Cntr=0.3,0.1

Type RM Length L Ch R = 1,45926,1004,1004,1004
BEGIN DESCRIPTION:
XS2973A
END DESCRIPTION:
XS GIS Cut Line= 4
      2800018.85      7074115.02      2799654.29      7073552.57
      2799487.62      7073432.77      2798821.77      7072959.39
#Sta/Elev= 30
  4255.6  492.43  4454.0  491.50  4511.4  489.28  4599.9  487.57  4677.5  485.63
  4750.0  486.25  4837.7  483.80  4920.5  485.70  4930.7  486.12  4966.3  483.98
  4987.2  475.23  4990.5  474.65  4991.4  473.85  5000.2  473.85  5001.0  474.65
  5001.9  480.25  5010.5  484.55  5016.6  485.23  5174.3  487.02  5259.9  483.13
  5325.1  485.82  5339.9  485.52  5390.3  483.02  5396.5  481.66  5411.2  483.04
  5503.4  486.45  5568.6  486.42  5587.8  487.57  5752.4  491.37  5948.1  497.83
#Mann=6,-1,0
  4255.6    0.05       0  4920.5    0.12       0  4990.5    0.07       0
  5001.0    0.12       0  5174.3    0.16       0  5752.4    0.05       0
Bank Sta=4599.9,5587.8
Exp/Cntr=0.3,0.1

Type RM Length L Ch R = 1,44922,514,514,514
BEGIN DESCRIPTION:
SCHOOLEY CREEK 39.0
END DESCRIPTION:
XS GIS Cut Line= 3
      2799975.00      7073974.99      2799775.99      7073080.00
      2799574.99      7072574.98
#Sta/Elev= 30
  3973.4  494.14  4268.8  486.64  4317.8  485.69  4495.8  485.47  4545.6  486.25
  4607.3  485.14  4659.8  486.18  4670.0  485.98  4690.0  483.70  4700.7  482.79
  4752.0  482.44  4778.6  483.83  4909.1  484.56  4971.0  483.28  4981.7  475.19
  4982.0  474.00  4982.9  473.20  4991.8  473.20  4992.6  474.00  4992.7  477.66
  5003.3  479.21  5011.6  484.03  5057.1  484.19  5083.3  486.64  5100.6  489.44
  5132.4  492.86  5183.5  495.98  5304.6  500.45  5365.0  499.55  5433.8  500.74
#Mann=6,-1,0
  3973.4    0.05       0  4607.3    0.16       0  4690.0    0.12       0
  4982.0    0.07       0  4992.6    0.12       0  5183.5    0.05       0
Bank Sta=4268.8,5083.3
Exp/Cntr=0.3,0.1

Type RM Length L Ch R = 1,44408,395,395,395
BEGIN DESCRIPTION:
XS2974A
END DESCRIPTION:
XS GIS Cut Line= 4
      2800190.75      7074016.13      2800091.79      7073010.90
      2800060.54      7072917.15      2799805.35      7072661.96
#Sta/Elev= 30
  3957.0  493.07  4065.2  490.02  4219.4  486.88  4401.0  485.74  4602.3  485.49
  4641.4  484.91  4671.6  485.99  4711.8  484.47  4752.0  484.47  4812.2  482.32
  4833.7  482.47  4872.5  482.01  4880.4  481.08  4892.6  481.02  4970.4  483.48
  4975.7  482.30  4989.1  473.36  4989.9  472.56  4998.8  472.56  4999.7  473.36
  5015.5  481.65  5026.0  483.70  5033.6  484.28  5091.0  484.76  5109.8  485.74
  5135.0  488.44  5170.3  489.35  5201.2  491.26  5318.8  497.03  5426.8  498.51
#Mann=7,-1,0
  3957.0    0.05       0  4602.3    0.16       0  4833.7    0.12       0
  4989.1    0.07       0  4999.7    0.12       0  5091.0    0.16       0
  5201.2    0.05       0
Bank Sta=4401,5109.8
Exp/Cntr=0.3,0.1

Type RM Length L Ch R = 1,44013,1474,1474,1474
BEGIN DESCRIPTION:
SCHOOLEY CREEK 38.0
END DESCRIPTION:
XS GIS Cut Line= 3
      2800852.19      7073724.41      2800340.40      7072976.32
      2799724.97      7072524.98
#Sta/Elev= 30
  4093.6  490.54  4362.8  485.29  4480.8  483.97  4507.9  483.15  4529.1  479.65
  4552.6  483.10  4594.5  483.68  4854.6  482.24  4875.6  479.02  4892.0  481.48
  4977.2  482.64  4992.5  472.75  4993.3  471.95  5003.1  472.75  5005.6  479.06
  5011.8  481.36  5032.6  482.69  5141.4  482.20  5147.6  484.18  5162.3  482.56
  5298.1  482.96  5313.1  485.29  5319.0  489.95  5334.7  491.57  5340.6  490.63
  5348.3  488.37  5354.5  491.03  5383.8  493.32  5590.7  499.52  5763.2  499.88
#Mann=7,-1,0
  4093.6    0.05       0  4480.8    0.16       0  4892.0    0.12       0
  4992.5    0.07       0  5003.1    0.12       0  5334.7    0.16       0
  5340.6    0.05       0
Bank Sta=4362.8,5313.1
Exp/Cntr=0.3,0.1

Type RM Length L Ch R = 1,42539,1311,1311,1311
BEGIN DESCRIPTION:
XS2975A
END DESCRIPTION:
XS GIS Cut Line= 3
      2801393.85      7073505.66      2800664.71      7072656.73
      2800435.51      7072380.65
#Sta/Elev= 30
  3811.1  496.71  4250.0  483.89  4261.5  483.60  4434.5  480.29  4456.5  477.50
  4477.3  480.17  4491.6  476.47  4498.2  480.42  4505.9  475.82  4512.4  478.59
  4520.1  474.41  4526.7  480.31  4534.4  477.97  4562.9  480.92  4796.5  482.09
  4887.8  478.94  4923.7  480.96  4966.9  481.62  4987.7  474.78  4990.2  471.53
  4991.1  470.73  5000.8  471.53  5009.9  480.91  5018.1  481.56  5088.0  483.62
  5094.5  478.17  5101.4  478.98  5107.8  483.89  5147.8  488.28  5289.0  488.87
#Mann=9,-1,0
  3811.1    0.05       0  4261.5    0.16       0  4796.5    0.12       0
  4887.8    0.16       0  4923.7    0.12       0  4990.2    0.07       0
  5000.8    0.12       0  5018.1    0.16       0  5147.8    0.05       0
Bank Sta=4250,5107.8
Exp/Cntr=0.3,0.1

Type RM Length L Ch R = 1,41228,375,375,375
BEGIN DESCRIPTION:
XS2976A
END DESCRIPTION:
XS GIS Cut Line= 3
      2801680.30      7073010.87      2801222.00      7072552.57
      2800534.55      7072385.91
#Sta/Elev= 30
  4326.8  505.24  4454.9  499.65  4483.2  496.60  4504.4  496.61  4540.8  494.63
  4603.4  490.43  4681.2  483.22  4714.8  482.15  4781.7  480.26  4850.9  479.00
  4900.4  480.93  4964.0  479.38  4969.7  478.29  4981.4  478.12  4986.6  470.96
  4987.1  469.09  4987.9  468.29  4997.0  468.29  4997.8  469.09  5002.7  469.32
  5013.0  472.59  5023.2  480.42  5032.5  480.34  5136.5  480.30  5187.9  479.27
  5467.3  482.15  5503.4  484.49  5535.1  486.43  5618.7  488.52  5682.3  488.09
#Mann=7,-1,0
  4326.8    0.08       0  4540.8    0.16       0  4781.7    0.12       0
  4987.1    0.07       0  4997.8    0.12       0  5032.5    0.16       0
  5503.4    0.05       0
Bank Sta=4714.8,5467.3
Exp/Cntr=0.3,0.1

Type RM Length L Ch R = 1,40853,786,786,786
BEGIN DESCRIPTION:
XS2979A
END DESCRIPTION:
XS GIS Cut Line= 3
      2801659.48      7072844.21      2801320.96      7072286.94
      2800659.78      7071823.60
#Sta/Elev= 30
  4325.9  499.94  4451.0  494.06  4575.9  487.76  4628.2  481.95  4672.4  481.68
  4707.8  480.29  4771.7  478.53  4802.6  480.65  4831.6  477.95  4961.6  479.33
  4976.1  478.48  4984.6  472.38  4985.3  469.17  4986.1  468.37  4996.0  469.17
  4997.4  472.13  5005.5  478.38  5011.6  479.78  5056.0  478.48  5274.6  480.04
  5284.8  479.98  5321.1  481.30  5461.2  478.99  5631.6  478.46  5637.6  478.08
  5644.6  476.52  5653.1  481.68  5666.3  491.30  5672.4  491.99  5785.3  494.33
#Mann=11,-1,0
  4325.9    0.08       0  4451.0    0.16       0  4707.8    0.12       0
  4831.6    0.16       0  4985.3    0.07       0  4996.0    0.16       0
  5274.6    0.05       0  5284.8    0.16       0  5461.2    0.12       0
  5631.6    0.16       0  5637.6    0.05       0
Bank Sta=4672.4,5653.1
Exp/Cntr=0.3,0.1

Type RM Length L Ch R = 1,40067,171,171,171
BEGIN DESCRIPTION:
XS2977A
END DESCRIPTION:
XS GIS Cut Line= 6
      2801675.13      7072703.63      2801586.58      7072224.44
      2801492.83      7071990.07      2801352.21      7071818.19
      2801201.17      7071724.44      2800883.66      7071609.93
#Sta/Elev= 30
  3860.6  495.97  3920.2  494.30  3948.8  490.60  3971.1  490.23  3997.7  492.74
  4062.6  490.33  4128.4  490.80  4251.6  486.70  4351.8  483.29  4388.0  483.13
  4495.6  480.74  4617.9  479.58  4776.3  477.56  4794.3  479.13  4814.7  478.11
  4902.5  477.79  4974.3  476.50  4983.8  474.67  4989.5  469.57  4990.3  468.77
  5000.4  469.57  5005.8  473.39  5015.8  475.18  5043.3  476.55  5054.1  480.74
  5074.0  483.62  5120.2  484.84  5314.3  494.01  5329.1  494.47  5337.7  494.13
#Mann=17,-1,0
  3860.6    0.08       0  3948.8    0.16       0  4128.4    0.08       0
  4251.6    0.16       0  4351.8    0.08       0  4388.0    0.16       0
  4617.9    0.05       0  4776.3    0.12       0  4814.7    0.05       0
  4902.5    0.16       0  4989.5    0.07       0  5000.4    0.16       0
  5005.8    0.05       0  5015.8    0.08       0  5120.2    0.05       0
  5314.3    0.08       0  5329.1    0.05       0
Bank Sta=4495.6,5054.1
Exp/Cntr=0.3,0.1

Type RM Length L Ch R = 1,39896,791,791,791
BEGIN DESCRIPTION:
XS2978A
END DESCRIPTION:
XS GIS Cut Line= 6
      2801820.96      7072578.62      2801669.92      7072036.94
      2801456.37      7071771.32      2801248.04      7071604.65
      2801169.92      7071547.36      2800836.58      7071349.44
#Sta/Elev= 30
  3753.7  500.10  3907.1  497.81  3960.9  494.56  4019.6  491.61  4121.8  490.33
  4301.0  484.28  4448.4  479.83  4564.1  479.23  4581.1  479.06  4659.1  478.06
  4888.5  478.34  4939.8  479.78  4961.9  474.24  4989.4  472.62  4991.9  468.35
  4992.7  467.55  5002.8  468.35  5018.3  470.50  5020.5  477.33  5033.5  478.88
  5049.1  479.12  5063.5  475.48  5084.4  480.58  5092.0  477.52  5094.3  479.06
  5097.8  481.34  5114.2  481.64  5142.6  482.35  5165.8  485.90  5408.2  493.91
#Mann=12,-1,0
  3753.7    0.05       0  3960.9    0.08       0  4019.6    0.05       0
  4121.8    0.08       0  4301.0    0.05       0  4564.1    0.16       0
  4659.1    0.05       0  4888.5    0.16       0  4991.9    0.04       0
  5002.8    0.16       0  5063.5    0.16       0  5114.2    0.05       0
Bank Sta=4581.1,5094.3
Exp/Cntr=0.3,0.1

Type RM Length L Ch R = 1,39105,684,684,684
BEGIN DESCRIPTION:
SCHOOLEY CREEK 33.0
END DESCRIPTION:
XS GIS Cut Line= 3
      2801975.03      7071525.03      2801475.00      7071075.00
      2800875.01      7071125.00
#Sta/Elev= 30
  4325.4  493.06  4424.5  485.69  4509.7  484.83  4573.5  478.90  4722.0  476.22
  4856.5  477.45  4870.7  473.65  4891.6  477.34  4941.6  477.36  4976.8  476.93
  4984.3  468.42  4989.3  467.41  4990.1  466.61  5000.2  467.41  5008.2  468.69
  5018.2  474.78  5038.3  477.60  5105.1  477.57  5138.6  478.50  5158.7  473.22
  5168.7  472.87  5188.8  473.69  5208.9  476.97  5244.2  477.12  5379.4  475.17
  5472.2  476.42  5485.2  478.90  5506.3  486.42  5519.9  493.59  5600.2  494.32
#Mann=8,-1,0
  4325.4    0.05       0  4941.6    0.12       0  4989.3    0.07       0
  5000.2    0.12       0  5105.1    0.05       0  5244.2    0.12       0
  5472.2    0.16       0  5506.3    0.05       0
Bank Sta=4573.5,5485.2
Exp/Cntr=0.3,0.1

Type RM Length L Ch R = 1,38421,782,782,782
BEGIN DESCRIPTION:
SCHOOLEY CREEK 32.0
END DESCRIPTION:
XS GIS Cut Line= 3
      2802274.98      7071474.97      2802025.00      7070925.00
      2801425.01      7070675.01
#Sta/Elev= 30
  4386.8  494.85  4452.7  495.16  4591.1  493.00  4628.4  493.41  4711.9  491.32
  4763.5  491.54  4786.6  490.61  4861.3  484.01  4921.2  481.44  4973.9  478.07
  4976.6  477.65  4982.1  470.23  4988.2  467.86  4994.7  467.42  4995.4  466.62
  5005.6  467.42  5012.6  475.15  5034.8  476.40  5066.7  475.31  5175.1  475.96
  5196.7  474.70  5218.4  476.04  5247.1  475.64  5327.1  475.26  5381.4  475.16
  5502.2  478.07  5565.1  481.58  5586.7  483.91  5597.0  486.55  5640.9  489.31
#Mann=7,-1,0
  4386.8    0.05       0  4921.2    0.12       0  4994.7    0.07       0
  5005.6    0.12       0  5247.1    0.16       0  5327.1    0.12       0
  5381.4    0.05       0
Bank Sta=4973.9,5502.2
Exp/Cntr=0.3,0.1

Type RM Length L Ch R = 1,37639,871,871,871
BEGIN DESCRIPTION:
XS2980A
END DESCRIPTION:
XS GIS Cut Line= 3
      2802623.04      7070781.74      2802326.17      7070516.11
      2801473.09      7070219.61
#Sta/Elev= 30
  4600.8  489.72  4667.7  488.03  4802.0  489.61  4965.3  485.21  4972.8  480.26
  4979.5  480.71  4982.0  476.51  4987.0  468.03  4991.1  465.77  4991.9  464.97
  5002.1  465.77  5011.0  466.01  5017.0  472.38  5032.2  474.43  5125.9  475.27
  5229.5  474.49  5243.9  469.34  5265.9  474.02  5275.7  469.79  5297.0  474.53
  5307.4  470.63  5317.5  470.72  5322.8  474.14  5328.6  474.60  5370.9  471.34
  5385.1  474.22  5542.0  473.77  5663.1  476.51  5796.2  480.61  5902.3  486.08
#Mann=7,-1,0
  4600.8    0.05       0  4802.0    0.16       0  4991.1    0.07       0
  5002.1    0.16       0  5125.9    0.12       0  5542.0    0.05       0
  5796.2    0.16       0
Bank Sta=4982,5663.1
Exp/Cntr=0.3,0.1

Type RM Length L Ch R = 1,36768,814,814,814
BEGIN DESCRIPTION:
SCHOOLEY CREEK 30.0
END DESCRIPTION:
XS GIS Cut Line= 3
      2802874.98      7070474.98      2802425.00      7070075.00
      2801524.95      7070075.00
#Sta/Elev= 30
  4472.2  488.65  4564.6  485.97  4826.3  483.00  4854.7  479.12  4875.7  480.02
  4911.6  484.27  4953.8  485.76  4958.9  481.00  4960.9  479.14  4967.6  484.12
  4971.3  475.68  4975.2  466.95  4981.9  473.36  4989.4  463.67  4996.1  465.63
  5010.3  463.83  5032.0  464.35  5033.2  463.18  5034.0  462.38  5044.2  463.18
  5076.8  463.32  5084.3  464.46  5104.3  473.08  5114.3  473.56  5474.3  472.80
  5580.6  473.97  5679.7  475.29  5689.7  475.68  5814.3  478.38  5974.3  487.41
#Mann=6,-1,0
  4472.2    0.05       0  4958.9    0.12       0  5033.2    0.07       0
  5044.2    0.12       0  5580.6    0.16       0  5679.7    0.05       0
Bank Sta=4971.3,5689.7
Exp/Cntr=0.3,0.1

Type RM Length L Ch R = 1,35954,470,470,470
BEGIN DESCRIPTION:
XS2981A
END DESCRIPTION:
XS GIS Cut Line= 5
      2803263.63      7069995.25      2802826.17      7069714.02
      2802597.00      7069714.02      2802268.87      7069521.32
      2801763.63      7069432.77
#Sta/Elev= 30
  3874.8  487.96  4017.9  483.17  4120.9  485.34  4171.6  484.23  4329.6  483.44
  4436.0  478.87  4486.0  482.22  4576.0  482.28  4632.1  479.52  4645.7  480.23
  4696.5  478.57  4712.5  474.91  4719.1  472.87  4733.6  471.89  4968.1  472.66
  4974.3  465.49  4991.9  459.95  4992.6  459.15  5003.0  459.95  5003.9  463.13
  5008.4  463.13  5012.9  460.19  5018.6  464.61  5028.8  465.91  5038.9  471.41
  5097.3  471.44  5143.2  474.91  5272.4  483.20  5473.0  490.81  5517.5  490.20
#Mann=6,-1,0
  3874.8    0.16       0  4171.6    0.05       0  4645.7    0.12       0
  4991.9    0.07       0  5003.0    0.12       0  5097.3    0.16       0
Bank Sta=4712.5,5143.2
Exp/Cntr=0.3,0.1

Type RM Length L Ch R = 1,35484,1100,1100,1100
BEGIN DESCRIPTION:
SCHOOLEY CREEK 28.0
END DESCRIPTION:
XS GIS Cut Line= 3
      2803475.00      7070025.00      2802518.83      7069186.36
      2801825.04      7069075.01
#Sta/Elev= 30
  3602.8  495.64  3733.0  489.72  3766.0  488.29  3801.6  486.06  4020.8  481.26
  4209.4  482.53  4311.2  481.43  4382.4  482.68  4509.5  482.07  4644.3  478.84
  4725.8  474.71  4766.2  473.91  4929.2  470.77  4976.3  472.02  4989.9  471.10
  5004.6  459.27  5005.3  458.47  5015.7  459.27  5020.3  466.65  5030.4  471.21
  5038.2  471.98  5141.8  470.90  5182.4  471.94  5198.4  473.91  5229.1  478.34
  5259.2  480.21  5353.0  486.91  5414.9  489.37  5526.7  489.11  5577.3  490.30
#Mann=8,-1,0
  3602.8    0.16       0  3733.0    0.05       0  3766.0    0.16       0
  4209.4    0.05       0  4725.8    0.12       0  5004.6    0.07       0
  5015.7    0.12       0  5259.2    0.05       0
Bank Sta=4766.2,5198.4
Exp/Cntr=0.3,0.1

Type RM Length L Ch R = 1,34384,741,741,741
BEGIN DESCRIPTION:
SCHOOLEY CREEK 27.0
END DESCRIPTION:
XS GIS Cut Line= 3
      2803164.74      7068823.41      2802325.00      7068575.00
      2802039.88      7068656.68
#Sta/Elev= 30
  4136.6  485.38  4188.8  486.21  4255.3  484.91  4288.6  482.26  4293.8  482.97
  4313.6  481.01  4327.3  480.88  4360.3  480.17  4459.6  475.08  4496.8  471.32
  4503.8  469.15  4531.9  468.22  4543.0  469.45  4595.2  468.76  4626.5  470.06
  4682.4  469.17  4787.9  468.95  4957.2  470.45  4970.6  468.41  4987.8  459.37
  4990.1  458.25  4990.8  457.45  5000.5  457.45  5001.2  458.25  5001.9  460.73
  5009.7  470.71  5018.8  471.32  5089.7  474.84  5230.8  484.69  5308.9  486.19
#Mann=8,-1,0
  4136.6    0.16       0  4327.3    0.12       0  4682.4    0.05       0
  4787.9    0.12       0  4987.8    0.16       0  4990.1    0.07       0
  5001.2    0.16       0  5089.7    0.05       0
Bank Sta=4496.8,5018.8
Exp/Cntr=0.3,0.1

Type RM Length L Ch R = 1,33643,470,470,470
BEGIN DESCRIPTION:
SCHOOLEY CREEK 26.0
END DESCRIPTION:
XS GIS Cut Line= 3
      2803174.98      7068324.99      2802625.00      7068025.00
      2802024.95      7067975.00
#Sta/Elev= 30
  4398.3  486.31  4539.4  477.80  4575.3  472.11  4598.1  470.69  4619.0  467.60
  4635.1  467.93  4640.8  465.55  4656.9  467.68  4662.6  465.03  4700.6  466.94
  4706.3  464.46  4728.6  464.07  4774.2  465.48  4782.2  466.21  4787.9  469.41
  4797.0  469.69  4967.3  469.11  4973.0  468.22  4989.2  461.19  4989.3  457.11
  4990.0  456.31  5000.5  457.11  5011.0  457.31  5016.7  460.10  5032.2  462.36
  5054.9  468.64  5145.2  468.25  5231.4  470.69  5416.1  475.74  5626.9  486.93
#Mann=5,-1,0
  4398.3    0.16       0  4539.4    0.12       0  4989.3    0.07       0
  5000.5    0.12       0  5032.2    0.05       0
Bank Sta=4598.1,5231.4
Exp/Cntr=0.3,0.1

Type RM Length L Ch R = 1,33173,1087,1087,1087
BEGIN DESCRIPTION:
XS2982A
END DESCRIPTION:
XS GIS Cut Line= 3
      2803461.63      7067911.96      2802940.75      7067656.73
      2802316.75      7067609.93
#Sta/Elev= 30
  4363.5  484.33  4439.7  483.53  4507.2  480.12  4604.7  473.44  4687.0  470.26
  4697.4  469.98  4816.3  467.63  4827.8  468.36  4872.8  466.20  4969.4  468.22
  4979.4  464.10  4983.8  455.85  4984.5  455.05  4994.4  455.05  4995.1  455.85
  4999.5  457.28  5009.5  463.76  5019.5  467.64  5029.0  468.49  5069.6  467.40
  5159.9  467.00  5166.1  466.00  5171.1  463.12  5180.0  466.74  5223.2  466.97
  5270.2  467.52  5342.5  470.26  5435.2  473.71  5520.9  478.61  5569.3  480.36
#Mann=5,-1,0
  4363.5    0.16       0  4697.4    0.12       0  4983.8    0.07       0
  4995.1    0.12       0  5223.2    0.05       0
Bank Sta=4687,5342.5
Exp/Cntr=0.3,0.1

Type RM Length L Ch R = 1,32086,1145,1145,1145
BEGIN DESCRIPTION:
SCHOOLEY CREEK 24.0
END DESCRIPTION:
XS GIS Cut Line= 3
      2803725.03      7067325.01      2803175.00      7067075.00
      2802525.00      7067025.00
#Sta/Elev= 30
  4409.0  484.18  4538.6  483.62  4579.2  482.57  4628.7  479.98  4686.9  475.67
  4792.0  469.00  4808.9  467.87  4892.4  465.24  4901.1  466.43  4958.3  466.46
  4969.2  465.11  4975.8  463.05  4991.2  456.87  4993.3  454.44  4994.0  453.64
  5003.9  453.64  5004.6  454.44  5010.4  462.07  5015.7  462.07  5023.2  466.15
  5053.3  465.93  5123.5  467.16  5163.6  465.74  5208.5  466.42  5314.1  466.67
  5470.9  469.00  5554.8  472.31  5584.9  475.56  5594.9  477.35  5665.1  481.93
#Mann=6,-1,0
  4409.0    0.05       0  4579.2    0.16       0  4686.9    0.12       0
  4993.3    0.07       0  5004.6    0.12       0  5208.5    0.05       0
Bank Sta=4792,5470.9
Exp/Cntr=0.3,0.1

Type RM Length L Ch R = 1,30941,1152,1152,1152
BEGIN DESCRIPTION:
XS2983A
END DESCRIPTION:
XS GIS Cut Line= 3
      2803727.18      7066630.69      2803133.46      7066547.36
      2802722.03      7066542.15
#Sta/Elev= 30
  4336.4  480.62  4413.8  478.06  4475.6  473.61  4485.1  472.58  4588.5  467.56
  4699.1  464.54  4793.0  464.27  4803.1  463.89  4813.2  461.95  4823.3  464.02
  4863.7  465.17  4873.8  464.47  4913.0  465.40  4978.0  463.95  4984.4  462.95
  4994.4  454.05  4998.7  453.55  4999.4  452.75  5009.5  452.75  5010.1  453.55
  5014.4  459.16  5024.4  464.91  5077.0  464.50  5144.4  465.45  5203.8  467.56
  5224.4  468.17  5244.4  470.07  5254.4  469.77  5274.4  472.13  5347.4  476.98
#Mann=6,-1,0
  4336.4    0.05       0  4475.6    0.12       0  4978.0    0.16       0
  4998.7    0.07       0  5010.1    0.16       0  5077.0    0.05       0
Bank Sta=4588.5,5203.8
Exp/Cntr=0.3,0.1

Type RM Length L Ch R = 1,29789,762,762,762
BEGIN DESCRIPTION:
XS2984A
END DESCRIPTION:
XS GIS Cut Line= 3
      2803695.97      7066391.12      2803279.29      7066156.73
      2802608.67      7066156.73
#Sta/Elev= 30
  4497.2  479.70  4555.3  480.01  4642.0  476.60  4657.9  476.12  4663.7  476.52
  4796.6  469.19  4842.7  467.77  4863.2  466.78  4912.3  466.75  4929.2  465.71
  4971.5  463.60  4974.9  460.50  4979.9  460.50  4983.9  453.47  4984.5  452.67
  4994.6  452.67  4995.3  453.47  4999.6  453.93  5019.6  462.67  5029.6  463.64
  5068.1  463.58  5154.0  463.28  5209.6  462.49  5239.6  463.38  5279.6  464.07
  5359.6  463.37  5459.1  465.71  5539.6  469.26  5579.6  472.13  5645.9  475.56
#Mann=7,-1,0
  4497.2    0.05       0  4842.7    0.12       0  4983.9    0.07       0
  4995.3    0.12       0  5068.1    0.16       0  5154.0    0.07       0
  5239.6    0.05       0
Bank Sta=4929.2,5459.1
Exp/Cntr=0.3,0.1

Type RM Length L Ch R = 1,29027,546,546,546
BEGIN DESCRIPTION:
SCHOOLEY CREEK 21.0
END DESCRIPTION:
XS GIS Cut Line= 3
      2803775.04      7065925.02      2803362.62      7065693.19
      2802425.00      7065875.00
#Sta/Elev= 30
  4511.0  479.05  4746.0  475.73  4917.8  471.84  4972.9  470.94  4984.1  469.81
  4986.9  465.36  4991.9  457.32  4996.4  453.58  4997.0  452.78  5007.2  452.78
  5007.8  453.58  5012.2  455.10  5018.6  461.34  5038.3  462.41  5057.4  462.16
  5134.5  461.45  5195.6  462.43  5277.1  461.06  5334.1  462.74  5379.0  461.51
  5419.7  462.34  5450.3  461.31  5531.7  461.44  5597.8  462.56  5656.2  465.36
  5758.1  471.08  5776.2  473.69  5796.6  473.27  5856.5  478.37  5939.2  483.22
#Mann=6,-1,0
  4511.0    0.05       0  4917.8    0.12       0  4996.4    0.07       0
  5007.8    0.12       0  5038.3    0.07       0  5057.4    0.05       0
Bank Sta=4986.9,5656.2
Exp/Cntr=0.3,0.1

Type RM Length L Ch R = 1,28481,161,161,161
BEGIN DESCRIPTION:
XS2985A
END DESCRIPTION:
XS GIS Cut Line= 3
      2803862.66      7065432.79      2803388.67      7065208.82
      2802728.60      7064891.78
#Sta/Elev= 30
  4452.4  473.77  4531.0  471.41  4555.8  471.99  4576.5  472.66  4673.1  468.82
  4721.5  465.20  4748.4  463.87  4764.1  464.37  4870.6  462.20  4981.5  460.33
  4997.2  452.03  4997.8  451.23  5008.0  451.23  5008.7  452.03  5014.0  457.64
  5025.4  456.84  5042.5  460.60  5059.1  461.38  5132.6  460.52  5223.6  459.76
  5268.9  460.95  5291.3  459.10  5365.0  460.86  5415.8  459.44  5478.2  461.20
  5525.2  463.91  5549.0  465.20  5614.6  469.23  5670.4  473.98  5708.9  475.69
#Mann=9,-1,0
  4452.4    0.05       0  4555.8    0.08       0  4870.6    0.12       0
  4997.2    0.07       0  5008.7    0.12       0  5059.1    0.08       0
  5132.6    0.12       0  5525.2    0.08       0  5614.6    0.12       0
Bank Sta=4721.5,5549
Exp/Cntr=0.3,0.1

Type RM Length L Ch R = 1,28320,704,704,704
BEGIN DESCRIPTION:
XS2986A
END DESCRIPTION:
XS GIS Cut Line= 3
      2803930.32      7065245.27      2803529.29      7065099.44
      2802838.31      7064772.13
#Sta/Elev= 30
  4490.9  470.67  4507.5  471.08  4528.9  471.55  4595.9  472.52  4603.0  471.57
  4613.8  465.18  4621.1  459.13  4626.5  458.20  4925.9  460.88  4977.7  460.40
  4984.8  458.12  4994.1  450.74  4994.7  449.94  5005.6  450.74  5022.0  460.76
  5034.3  460.94  5093.2  460.82  5142.7  460.81  5172.3  458.06  5177.8  459.88
  5195.0  456.08  5210.1  457.17  5217.8  460.68  5251.1  459.83  5333.7  460.14
  5359.5  461.23  5467.9  463.73  5491.9  465.18  5574.2  469.78  5682.2  476.47
#Mann=14,-1,0
  4490.9    0.08       0  4507.5    0.05       0  4528.9    0.12       0
  4925.9    0.05       0  4994.1    0.04       0  5005.6    0.05       0
  5034.3    0.08       0  5093.2    0.12       0  5142.7    0.05       0
  5251.1    0.08       0  5333.7    0.12       0  5359.5    0.05       0
  5467.9    0.08       0  5574.2    0.12       0
Bank Sta=4613.8,5491.9
Exp/Cntr=0.3,0.1

Type RM Length L Ch R = 1,27616,1857,1857,1857
BEGIN DESCRIPTION:
XS2987A
END DESCRIPTION:
XS GIS Cut Line= 4
      2804190.72      7065177.53      2804013.67      7064896.32
      2803919.92      7064724.44      2803081.36      7064422.35
#Sta/Elev= 30
  4679.6  472.61  4790.1  473.05  4830.7  472.72  4851.9  469.81  4940.2  466.86
  4958.1  465.12  4976.7  463.43  4989.8  451.56  4992.1  450.81  4992.8  450.01
  5003.6  450.81  5003.8  453.10  5009.7  459.13  5011.0  459.13  5019.3  460.36
  5128.5  460.37  5373.0  458.10  5521.2  459.13  5571.9  457.12  5633.3  458.78
  5744.4  458.99  5756.1  456.55  5776.2  458.25  5862.8  460.34  5943.7  465.12
  5991.0  467.29  6041.8  472.71  6047.1  471.43  6072.5  475.03  6099.0  476.24
#Mann=6,-1,0
  4679.6    0.05       0  4790.1    0.16       0  4992.1    0.07       0
  5003.6    0.16       0  5011.0    0.12       0  5862.8    0.16       0
Bank Sta=4958.1,5943.7
Exp/Cntr=0.3,0.1

Type RM Length L Ch R = 1,25759,965,965,965
BEGIN DESCRIPTION:
XS2988A
END DESCRIPTION:
XS GIS Cut Line= 3
      2804711.61      7064177.57      2804305.33      7064089.02
      2803139.31      7064266.01
#Sta/Elev= 30
  4581.5  475.71  4629.2  474.28  4806.6  473.51  4864.6  472.00  4884.8  470.33
  4948.7  467.03  4968.9  464.99  4977.2  463.84  4986.8  448.87  4987.4  448.07
  4997.8  448.07  4998.4  448.87  5003.3  452.37  5008.3  452.40  5017.9  458.17
  5108.9  457.02  5280.9  457.34  5341.8  456.18  5405.5  457.76  5554.0  457.77
  5614.6  456.79  5624.8  455.06  5634.9  456.84  5655.1  458.13  5725.9  457.12
  5887.7  459.07  5992.6  464.99  5997.3  465.28  6120.4  473.32  6176.7  474.60
#Mann=5,-1,0
  4581.5    0.16       0  4884.8    0.12       0  4986.8    0.07       0
  4998.4    0.12       0  5997.3    0.16       0
Bank Sta=4968.9,5992.6
Exp/Cntr=0.3,0.1

Type RM Length L Ch R = 1,24794,768,768,768
BEGIN DESCRIPTION:
XS2989A
END DESCRIPTION:
XS GIS Cut Line= 3
      2804794.88      7063474.44      2804461.58      7063458.82
      2803139.35      7064125.14
#Sta/Elev= 30
  4669.8  475.77  4785.5  472.97  4935.1  464.97  4960.0  457.03  4976.6  454.71
  4981.6  456.52  4999.9  447.41  5000.5  446.61  5011.5  447.41  5022.0  456.44
  5028.0  456.57  5206.4  454.31  5585.7  455.86  5615.5  453.56  5624.7  455.89
  5892.4  457.60  5920.3  457.01  5929.1  453.99  5951.5  457.79  5987.2  455.00
  6018.7  457.58  6041.0  454.41  6054.2  458.28  6098.8  458.51  6115.5  455.31
  6134.7  458.49  6279.6  461.27  6386.7  464.97  6424.2  465.62  6484.1  467.77
#Mann=7,-1,0
  4669.8    0.16       0  4785.5    0.12       0  4999.9    0.07       0
  5011.5    0.12       0  6134.7    0.16       0  6279.6    0.12       0
  6424.2    0.16       0
Bank Sta=4935.1,6386.7
Exp/Cntr=0.3,0.1
