--- UNT 047 in LFCCL Watershed.prj (project) ---

Proj Title=UNT 047 in LFCCL Watershed Base Level Engineering
Current Plan=p01
Default Exp/Contr=0.3,0.1
English Units
Geom File=g01
Flow File=f01
Plan File=p01
BEGIN DESCRIPTION:
UNT 047 in LFCCL Watershed
END DESCRIPTION:

--- UNT 047 in LFCCL Watershed.p01 (plan) ---

Plan Title=Multiple Run
Short Identifier=Multiple
Geom File=g01
Flow File=f01
Subcritical Flow
K Sum by GR= 0
Std Step Tol= 0.01
Critical Tol= 0.01
Num of Std Step Trials= 20
Max Error Tol= 0.3
Flow Tol Ratio= 0.001
Split Flow NTrial= 30
Split Flow Tol= 0.02
Split Flow Ratio= 0.02
Log Output Level= 0
Friction Slope Method= 1
Unsteady Friction Slope Method= 2
Unsteady Bridges Friction Slope Method= 1
Parabolic Critical Depth
Global Vel Dist=  1 , 1 , 1
Global Log Level= 0
CheckData=True
Encroach Param= -1, 0, 0, 0
BEGIN DESCRIPTION:
Multiple Run
END DESCRIPTION:

--- UNT 047 in LFCCL Watershed.f01 (steady flow) ---

Flow Title=Multiple
Number of Profiles=7
Profile Names=10-year,25-year,50-year,1pct_min,100-year,1pct_plu,500-year
River Rch & RM= UNT 047 in LFCCL,Reach-1,16084
     269     341     397     230     459     916     615
River Rch & RM= UNT 047 in LFCCL,Reach-1,11020
     484     638     760     451     899    1795    1260
River Rch & RM= UNT 047 in LFCCL,Reach-1,7821
     620     827     995     594    1185    2365    1686
River Rch & RM= UNT 047 in LFCCL,Reach-1,2992
     905    1234    1505     911    1817    3625    2654
Boundary for River Rch & Prof#=UNT 047 in LFCCL,Reach-1,1
Up Type=0
Dn Type=3
Dn Slope=0.005
Boundary for River Rch & Prof#=UNT 047 in LFCCL,Reach-1,2
Up Type=0
Dn Type=3
Dn Slope=0.005
Boundary for River Rch & Prof#=UNT 047 in LFCCL,Reach-1,3
Up Type=0
Dn Type=3
Dn Slope=0.005
Boundary for River Rch & Prof#=UNT 047 in LFCCL,Reach-1,4
Up Type=0
Dn Type=3
Dn Slope=0.005
Boundary for River Rch & Prof#=UNT 047 in LFCCL,Reach-1,5
Up Type=0
Dn Type=3
Dn Slope=0.005
Boundary for River Rch & Prof#=UNT 047 in LFCCL,Reach-1,6
Up Type=0
Dn Type=3
Dn Slope=0.005
Boundary for River Rch & Prof#=UNT 047 in LFCCL,Reach-1,7
Up Type=0
Dn Type=3
Dn Slope=0.005

--- UNT 047 in LFCCL Watershed.g01 (geometry) ---

Geom Title=Existing Conditions

River Reach=UNT 047 in LFCCL,Reach-1
Reach XY= 30
      2801916.60      7047750.27      2802044.73      7047299.58
      2801678.03      7046335.16      2801803.69      7045725.90
      2801429.04      7044835.69      2801830.60      7044592.66
      2801740.70      7044430.09      2802043.02      7042946.44
      2801392.99      7042346.88      2801231.82      7041522.20
      2800755.11      7040995.60      2801254.11      7040024.41
      2801493.06      7039874.95      2801382.94      7039690.07
      2801532.26      7039618.57      2801428.91      7039407.04
      2801554.18      7039346.72      2801299.20      7039139.13
      2801279.68      7038741.37      2801369.50      7038447.05
      2801553.18      7038414.87      2801447.01      7038291.32
      2801611.52      7037716.05      2801234.69      7037292.65
      2800944.48      7037275.68      2800925.19      7036892.55
      2800456.58      7037015.62      2800494.52      7036811.17
      2800337.51      7036928.43      2800095.59      7036700.71

Type RM Length L Ch R = 1,16084,305,305,305
BEGIN DESCRIPTION:
UNT 047 in LFCCL Watershed 31.0
END DESCRIPTION:
XS GIS Cut Line= 3
      2802166.00      7047752.49      2801980.66      7047628.93
      2801691.51      7047673.42
#Sta/Elev= 30
  4783.1  484.31  4788.9  484.06  4819.0  484.18  4855.1  483.49  4868.4  483.65
  4876.1  483.40  4882.1  484.12  4891.1  483.99  4897.1  483.06  4905.0  482.44
  4918.1  481.87  4933.2  481.65  4969.2  482.07  4976.6  481.40  4996.3  481.16
  4996.8  480.36  5001.8  480.36  5002.3  481.16  5009.7  481.49  5014.7  481.36
  5066.0  482.44  5083.0  483.24  5102.6  482.94  5141.2  483.34  5146.3  483.21
  5183.6  483.88  5234.2  483.96  5272.7  484.48  5277.8  484.81  5298.4  484.78
#Mann=3,-1,0
  4783.1    0.05       0  4996.3    0.03       0  5002.3    0.05       0
Bank Sta=4905,5066
Exp/Cntr=0.3,0.1

Type RM Length L Ch R = 1,15779,32,32,32
BEGIN DESCRIPTION:
XS3241A
END DESCRIPTION:
XS GIS Cut Line= 6
      2802203.04      7047700.57      2802109.15      7047495.50
      2802064.68      7047344.77      2801983.13      7047359.59
      2801978.19      7047438.66      2801780.54      7047614.08
#Sta/Elev= 30
  4599.1  484.03  4660.2  483.81  4671.2  484.43  4693.2  482.85  4722.1  482.03
  4737.2  481.52  4769.6  481.72  4781.2  481.37  4803.6  482.22  4823.6  480.91
  4874.2  480.75  4874.7  479.95  4879.7  479.95  4880.2  480.75  4954.8  481.36
  5082.8  481.48  5112.8  481.14  5132.9  481.81  5146.6  481.68  5153.1  482.90
  5160.7  483.57  5167.3  483.39  5174.9  482.23  5189.1  481.05  5231.1  481.24
  5264.8  482.03  5323.7  482.65  5351.5  483.95  5365.5  483.44  5410.9  484.00
#Mann=3,-1,0
  4599.1    0.05       0  4874.2    0.03       0  4880.2    0.05       0
Bank Sta=4722.1,5264.8
Exp/Cntr=0.3,0.1

Type RM Length L Ch R = 1,15747,44,44,44
BEGIN DESCRIPTION:
XS3240A
END DESCRIPTION:
XS GIS Cut Line= 6
      2802195.62      7047606.66      2802114.10      7047349.71
      2802067.15      7047310.17      2801968.31      7047327.47
      2801946.07      7047413.95      2801779.01      7047544.16
#Sta/Elev= 30
  4640.3  483.89  4704.6  481.71  4745.8  481.43  4768.3  482.25  4798.2  481.09
  4817.1  483.18  4910.4  483.68  4925.2  483.01  4933.7  484.55  4939.9  483.46
  4944.7  484.93  4954.7  484.18  4970.5  485.28  5022.0  484.88  5030.6  484.62
  5034.3  483.59  5078.6  484.00  5087.3  484.90  5107.8  483.93  5148.5  484.63
  5172.6  483.29  5177.6  481.85  5192.0  480.88  5238.8  480.71  5239.3  479.91
  5244.3  479.91  5244.8  480.71  5312.2  481.71  5355.8  482.44  5380.6  483.99
#Mann=3,-1,0
  4640.3    0.05       0  5238.8    0.03       0  5244.8    0.05       0
Bank Sta=4704.6,5312.2
Exp/Cntr=0.3,0.1

Type RM Length L Ch R = 1,15703,65,65,65
BEGIN DESCRIPTION:
XS3239A
END DESCRIPTION:
XS GIS Cut Line= 3
      2802366.13      7047273.11      2802039.96      7047270.63
      2801750.88      7047275.58
#Sta/Elev= 30
  4672.3  482.97  4703.4  482.06  4713.4  481.92  4733.4  482.06  4753.4  481.84
  4773.4  481.88  4783.4  482.33  4793.4  482.10  4803.4  481.46  4823.4  480.73
  4843.4  480.70  4853.4  480.55  4863.4  480.18  4902.8  479.83  4905.2  479.80
  4933.4  479.54  4952.4  479.72  4973.4  480.19  4983.4  480.11  4998.5  479.45
  5023.4  479.09  5060.5  478.86  5061.0  478.06  5066.0  478.06  5066.5  478.86
  5103.5  479.56  5163.5  479.20  5201.5  479.80  5241.4  480.47  5287.6  481.25
#Mann=6,-1,0
  4672.3    0.05       0  4902.8    0.08       0  4952.4    0.05       0
  5060.5    0.03       0  5066.5    0.05       0  5241.4    0.08       0
Bank Sta=4905.2,5201.5
Exp/Cntr=0.3,0.1

Type RM Length L Ch R = 1,15638,188,188,188
BEGIN DESCRIPTION:
XS3242A
END DESCRIPTION:
XS GIS Cut Line= 4
      2802240.10      7047117.44      2802119.04      7047203.92
      2802005.37      7047213.80      2801713.81      7047203.92
#Sta/Elev= 30
  4743.5  481.49  4745.8  481.24  4774.3  481.43  4796.1  481.20  4846.5  480.09
  4867.4  480.59  4887.1  480.45  4904.2  479.97  4936.5  479.25  4951.5  478.68
  4962.0  478.17  4967.1  478.41  4973.6  477.31  4974.1  476.51  4979.1  476.51
  4979.6  477.31  5009.1  477.43  5026.8  478.02  5076.8  478.78  5115.2  479.04
  5120.2  478.61  5124.2  478.68  5156.8  479.13  5166.0  479.54  5176.8  480.19
  5186.8  480.43  5216.9  480.60  5236.9  481.16  5256.9  481.42  5298.1  481.64
#Mann=6,-1,0
  4743.5    0.05       0  4887.1    0.08       0  4904.2    0.05       0
  4973.6    0.03       0  4979.6    0.05       0  5166.0    0.08       0
Bank Sta=4951.5,5124.2
Exp/Cntr=0.3,0.1

Type RM Length L Ch R = 1,15450,174,174,174
BEGIN DESCRIPTION:
XS3243A
END DESCRIPTION:
XS GIS Cut Line= 3
      2802250.02      7047045.77      2801958.42      7047048.24
      2801671.74      7047045.77
#Sta/Elev= 30
  4705.8  480.95  4780.8  480.39  4800.8  480.03  4820.8  479.91  4840.8  479.42
  4870.8  479.40  4880.8  479.64  4890.8  479.50  4910.8  478.75  4930.8  478.48
  4949.8  477.72  4970.8  476.81  5007.8  476.01  5008.3  475.21  5013.3  475.21
  5013.8  476.01  5020.8  476.59  5030.8  476.42  5050.8  476.51  5060.8  476.76
  5070.8  477.51  5077.0  477.72  5110.8  477.76  5130.8  478.07  5160.8  478.82
  5170.8  479.49  5180.8  479.85  5200.8  479.67  5220.8  479.15  5284.1  480.09
#Mann=3,-1,0
  4705.8    0.05       0  5007.8    0.03       0  5013.8    0.05       0
Bank Sta=4949.8,5077
Exp/Cntr=0.3,0.1

Type RM Length L Ch R = 1,15276,171,171,171
BEGIN DESCRIPTION:
XS3244A
END DESCRIPTION:
XS GIS Cut Line= 3
      2802074.54      7046850.56      2801886.76      7046892.57
      2801624.87      7046954.33
#Sta/Elev= 30
  4807.3  480.41  4809.6  480.41  4827.3  479.40  4837.6  479.13  4851.7  479.11
  4858.1  478.86  4909.3  478.13  4943.7  477.38  4966.7  476.61  4987.1  475.91
  4992.2  475.95  4998.1  475.63  5011.8  475.42  5019.1  475.02  5019.6  474.22
  5024.6  474.22  5025.1  475.02  5034.8  475.42  5042.6  475.95  5063.2  476.04
  5072.0  476.64  5077.1  476.49  5080.1  476.61  5114.3  477.54  5124.8  478.62
  5145.4  478.42  5155.6  478.92  5166.9  478.61  5176.2  478.63  5268.8  479.56
#Mann=3,-1,0
  4807.3    0.05       0  5019.1    0.03       0  5025.1    0.05       0
Bank Sta=4966.7,5080.1
Exp/Cntr=0.3,0.1

Type RM Length L Ch R = 1,15105,164,164,164
BEGIN DESCRIPTION:
XS3245A
END DESCRIPTION:
XS GIS Cut Line= 3
      2802089.40      7046731.95      2801790.39      7046749.25
      2801563.01      7046783.85
#Sta/Elev= 30
  4706.7  479.58  4711.4  479.58  4721.1  479.86  4731.1  478.88  4741.2  478.48
  4771.2  478.13  4841.2  476.77  4846.2  476.87  4871.4  476.34  4891.4  476.28
  4901.4  476.09  4918.4  475.50  4951.5  474.63  4991.6  474.27  4998.4  473.82
  4998.9  473.02  5003.9  473.02  5004.4  473.82  5006.2  473.82  5008.9  474.16
  5054.0  475.50  5062.2  475.65  5092.6  476.83  5102.7  477.35  5112.8  477.59
  5133.0  477.34  5146.2  477.34  5193.7  477.77  5214.8  478.16  5236.2  478.26
#Mann=3,-1,0
  4706.7    0.05       0  4998.4    0.03       0  5004.4    0.05       0
Bank Sta=4918.4,5054
Exp/Cntr=0.3,0.1

Type RM Length L Ch R = 1,14941,227,227,227
BEGIN DESCRIPTION:
XS3246A
END DESCRIPTION:
XS GIS Cut Line= 3
      2802072.08      7046596.04      2801800.28      7046583.69
      2801616.79      7046620.39
#Sta/Elev= 30
  4722.6  479.58  4729.7  479.30  4829.8  477.63  4855.3  476.91  4860.3  476.99
  4909.9  475.59  4944.2  474.48  4969.9  473.54  4979.9  473.40  4989.8  473.09
  4994.7  473.09  4997.1  472.73  4997.6  471.93  5002.6  471.93  5003.1  472.73
  5010.3  473.47  5026.2  473.76  5031.3  474.03  5051.1  473.95  5071.5  474.25
  5078.5  474.48  5082.3  474.54  5091.8  475.01  5102.0  474.91  5133.3  475.70
  5142.8  476.00  5153.0  476.56  5163.2  476.71  5179.2  476.35  5181.8  476.53
#Mann=3,-1,0
  4722.6    0.05       0  4997.1    0.03       0  5003.1    0.05       0
Bank Sta=4944.2,5078.5
Exp/Cntr=0.3,0.1

Type RM Length L Ch R = 1,14714,207,207,207
BEGIN DESCRIPTION:
XS3247A
END DESCRIPTION:
XS GIS Cut Line= 3
      2802074.56      7046393.42      2801691.55      7046390.95
      2801481.56      7046452.71
#Sta/Elev= 30
  4612.1  479.17  4631.7  478.90  4681.7  478.73  4691.7  478.56  4711.7  477.92
  4751.7  477.27  4781.7  476.41  4811.7  475.93  4861.7  474.72  4903.6  473.24
  4921.7  472.55  4941.7  472.37  4961.7  472.52  4971.7  472.29  4995.1  472.28
  5001.9  471.65  5009.4  471.62  5009.9  470.82  5014.9  470.82  5015.4  471.62
  5022.4  473.07  5027.6  472.93  5031.0  473.24  5033.2  473.45  5043.6  473.75
  5047.9  474.15  5055.4  474.81  5066.2  475.60  5106.2  475.05  5214.0  476.94
#Mann=5,-1,0
  4612.1    0.05       0  5009.4    0.03       0  5015.4    0.05       0
  5047.9    0.16       0  5055.4    0.05       0
Bank Sta=4903.6,5031
Exp/Cntr=0.3,0.1

Type RM Length L Ch R = 1,14507,444,444,444
BEGIN DESCRIPTION:
XS3248A
END DESCRIPTION:
XS GIS Cut Line= 3
      2802089.37      7046213.03      2801713.79      7046193.27
      2801407.36      7046240.22
#Sta/Elev= 30
  4617.8  479.39  4622.5  479.39  4652.2  478.36  4671.4  477.93  4676.4  478.03
  4692.3  477.51  4782.4  475.91  4812.4  475.71  4866.7  474.45  4872.5  474.20
  4892.5  473.84  4936.5  472.29  4982.7  470.80  4993.9  471.01  4999.8  470.44
  5000.3  469.64  5005.3  469.64  5005.8  470.44  5012.9  471.01  5044.9  471.80
  5063.5  471.91  5070.7  472.29  5083.7  472.55  5112.3  473.86  5124.2  474.10
  5134.3  473.81  5144.4  473.80  5184.9  474.12  5265.8  475.81  5303.9  476.92
#Mann=5,-1,0
  4617.8    0.05       0  4999.8    0.03       0  5005.8    0.05       0
  5044.9    0.16       0  5112.3    0.05       0
Bank Sta=4936.5,5070.7
Exp/Cntr=0.3,0.1

Type RM Length L Ch R = 1,14063,50,50,50
BEGIN DESCRIPTION:
XS3249A
END DESCRIPTION:
XS GIS Cut Line= 5
      2802074.56      7045780.61      2801785.45      7045775.66
      2801698.96      7045775.66      2801614.95      7045812.73
      2801385.14      7045956.05
#Sta/Elev= 30
  4696.6  476.36  4726.2  475.78  4731.6  475.40  4756.2  475.21  4796.2  473.93
  4816.2  473.71  4836.2  473.02  4874.3  472.28  4886.2  472.10  4926.2  470.62
  4966.2  470.04  5077.1  470.49  5154.9  469.98  5155.4  469.18  5160.4  469.18
  5160.9  469.98  5167.0  470.11  5173.9  471.14  5179.7  470.84  5187.6  471.49
  5195.1  471.58  5201.0  470.94  5216.3  471.09  5222.9  471.55  5231.7  471.69
  5258.8  471.99  5268.2  471.79  5295.4  471.94  5315.5  472.28  5434.9  473.72
#Mann=3,-1,0
  4696.6    0.05       0  5154.9    0.03       0  5160.9    0.05       0
Bank Sta=4874.3,5315.5
Exp/Cntr=0.3,0.1

Type RM Length L Ch R = 1,14013,139,139,139
BEGIN DESCRIPTION:
XS3250A
END DESCRIPTION:
XS GIS Cut Line= 6
      2802091.88      7045746.01      2801760.74      7045736.13
      2801686.61      7045736.13      2801644.60      7045736.13
      2801582.83      7045770.72      2801349.07      7045915.90
#Sta/Elev= 30
  4710.6  477.33  4727.5  476.55  4867.5  473.08  4907.3  472.19  4912.3  472.37
  4929.5  471.82  4984.6  470.30  4985.1  469.50  4990.1  469.50  4990.6  470.30
  4997.6  470.33  5017.6  473.52  5027.6  474.30  5047.6  474.61  5062.0  474.45
  5119.3  474.80  5160.7  474.71  5164.6  474.36  5170.4  475.00  5186.3  474.69
  5192.0  474.93  5228.1  474.38  5260.5  473.52  5266.4  472.73  5296.9  471.61
  5344.9  471.82  5345.9  471.82  5412.9  472.24  5455.4  473.09  5504.0  473.67
#Mann=5,-1,0
  4710.6    0.05       0  4984.6    0.03       0  4990.6    0.05       0
  5062.0    0.16       0  5344.9    0.05       0
Bank Sta=4929.5,5345.9
Exp/Cntr=0.3,0.1

Type RM Length L Ch R = 1,13874,241,241,241
BEGIN DESCRIPTION:
XS3251A
END DESCRIPTION:
XS GIS Cut Line= 4
      2802079.46      7045664.47      2801713.79      7045664.47
      2801572.94      7045691.65      2801319.21      7045777.87
#Sta/Elev= 30
  4626.1  476.68  4710.6  474.57  4730.6  474.37  4740.6  474.61  4760.6  473.81
  4902.4  469.40  4944.2  468.26  4991.8  467.33  5000.7  466.56  5007.9  466.42
  5008.4  465.62  5013.4  465.62  5013.9  466.42  5018.5  467.25  5023.6  467.12
  5031.3  467.46  5051.6  467.80  5070.3  468.62  5075.4  469.16  5084.5  469.40
  5112.8  470.22  5125.1  470.91  5154.2  471.29  5160.3  471.17  5165.6  471.49
  5185.8  470.98  5223.1  471.11  5228.4  471.42  5249.2  471.29  5403.2  472.23
#Mann=5,-1,0
  4626.1    0.05       0  4944.2    0.16       0  5007.9    0.07       0
  5013.9    0.16       0  5125.1    0.05       0
Bank Sta=4902.4,5084.5
Exp/Cntr=0.3,0.1

Type RM Length L Ch R = 1,13633,373,373,373
BEGIN DESCRIPTION:
XS3252A
END DESCRIPTION:
XS GIS Cut Line= 3
      2801992.98      7045414.90      2801674.25      7045427.25
      2801303.56      7045506.33
#Sta/Elev= 30
  4667.3  475.30  4685.3  474.95  4695.3  475.11  4705.3  474.81  4715.3  474.00
  4765.4  472.57  4835.4  471.15  4855.4  471.15  4875.4  470.74  4905.5  469.96
  4945.5  468.23  4977.5  467.86  4983.4  467.25  5005.9  466.69  5013.2  466.12
  5013.7  465.32  5018.7  465.32  5019.2  466.12  5026.4  466.73  5044.6  466.79
  5049.7  467.32  5068.1  467.86  5159.3  469.65  5169.6  469.37  5230.9  469.33
  5237.6  468.86  5242.7  469.28  5271.8  468.48  5336.6  470.40  5365.3  470.51
#Mann=3,-1,0
  4667.3    0.05       0  5013.2    0.03       0  5019.2    0.05       0
Bank Sta=4977.5,5068.1
Exp/Cntr=0.3,0.1

Type RM Length L Ch R = 1,13260,269,269,269
BEGIN DESCRIPTION:
XS3253A
END DESCRIPTION:
XS GIS Cut Line= 3
      2801896.65      7045120.84      2801577.88      7045083.78
      2801231.95      7045172.73
#Sta/Elev= 30
  4656.7  474.79  4698.6  474.09  4727.4  472.91  4747.3  471.06  4752.3  471.12
  4769.1  469.92  4820.8  468.32  4840.9  467.68  4869.8  466.20  4889.9  466.92
  4914.0  465.30  4924.4  464.36  4981.7  464.43  4987.9  464.15  4988.4  463.35
  4993.4  463.35  4993.9  464.15  5004.5  464.79  5021.9  464.39  5040.1  465.47
  5052.9  465.77  5081.1  465.30  5126.7  466.21  5156.1  466.05  5167.4  466.48
  5203.0  466.81  5208.1  467.23  5238.5  467.40  5269.7  468.22  5334.8  469.07
#Mann=5,-1,0
  4656.7    0.05       0  4727.4    0.16       0  4820.8    0.05       0
  4987.9    0.03       0  4993.9    0.05       0
Bank Sta=4914,5081.1
Exp/Cntr=0.3,0.1

Type RM Length L Ch R = 1,12991,271,271,271
BEGIN DESCRIPTION:
XS3254A
END DESCRIPTION:
XS GIS Cut Line= 3
      2801733.56      7044950.34      2801429.62      7044881.15
      2801175.09      7044886.10
#Sta/Elev= 30
  4695.3  467.92  4724.6  466.50  4733.1  466.38  4827.0  464.34  4857.9  464.42
  4875.2  464.89  4880.3  464.48  4898.9  464.84  4973.6  463.17  5001.5  461.89
  5003.8  461.09  5004.3  460.29  5009.3  460.29  5009.8  461.09  5021.6  461.35
  5034.0  463.17  5041.6  464.43  5051.6  465.68  5071.7  466.35  5081.7  466.38
  5101.7  465.15  5111.7  465.25  5131.7  466.95  5141.7  467.52  5171.7  468.27
  5191.7  468.15  5201.7  468.59  5211.7  469.72  5231.7  468.74  5261.6  469.02
#Mann=4,-1,0
  4695.3    0.16       0  4733.1    0.05       0  5003.8    0.03       0
  5009.8    0.05       0
Bank Sta=4973.6,5034
Exp/Cntr=0.3,0.1

Type RM Length L Ch R = 1,12720,288,288,288
BEGIN DESCRIPTION:
XS3255A
END DESCRIPTION:
XS GIS Cut Line= 3
      2801812.66      7044873.76      2801595.18      7044700.77
      2801313.51      7044636.53
#Sta/Elev= 30
  4713.9  468.77  4733.0  467.87  4796.4  465.86  4817.9  465.15  4846.8  464.61
  4853.2  464.26  4861.2  464.29  4867.6  463.83  4917.6  462.12  4966.9  461.57
  4981.3  460.47  4991.8  460.26  4993.2  459.88  4993.7  459.08  4998.7  459.08
  4999.2  459.88  5002.2  460.35  5033.0  461.26  5040.5  462.12  5044.3  462.65
  5053.5  462.97  5082.2  463.24  5087.3  464.10  5125.2  464.30  5130.3  464.13
  5145.8  464.46  5178.4  465.48  5207.4  466.79  5258.7  467.51  5280.7  467.24
#Mann=4,-1,0
  4713.9    0.16       0  4796.4    0.05       0  4993.2    0.03       0
  4999.2    0.05       0
Bank Sta=4917.6,5040.5
Exp/Cntr=0.3,0.1

Type RM Length L Ch R = 1,12432,248,248,248
BEGIN DESCRIPTION:
XS3256A
END DESCRIPTION:
XS GIS Cut Line= 3
      2802039.99      7044723.02      2801842.28      7044589.57
      2801343.18      7044515.45
#Sta/Elev= 30
  4749.9  473.23  4784.3  471.84  4803.5  471.19  4831.8  469.61  4875.5  466.70
  4888.6  465.37  4902.5  464.40  4917.5  463.62  4953.5  462.60  4974.3  460.76
  4988.0  459.48  5002.9  459.12  5003.4  458.32  5008.4  458.32  5008.9  459.12
  5046.3  460.29  5057.5  460.09  5072.3  460.76  5086.8  461.48  5107.0  461.74
  5121.9  461.12  5137.3  461.88  5157.5  461.39  5191.3  461.56  5228.3  462.32
  5248.5  463.09  5309.2  464.01  5334.5  464.67  5440.6  466.39  5493.0  466.54
#Mann=5,-1,0
  4749.9    0.05       0  4784.3    0.16       0  4831.8    0.05       0
  5002.9    0.03       0  5008.9    0.05       0
Bank Sta=4974.3,5072.3
Exp/Cntr=0.3,0.1

Type RM Length L Ch R = 1,12184,218,218,218
BEGIN DESCRIPTION:
XS3257A
END DESCRIPTION:
XS GIS Cut Line= 3
      2802072.04      7044475.89      2801763.21      7044391.89
      2801511.21      7044396.83
#Sta/Elev= 30
  4676.5  467.20  4694.0  466.71  4714.9  465.51  4766.7  463.72  4797.8  462.10
  4813.3  461.61  4828.9  460.84  4860.0  460.66  4880.7  460.87  4887.7  461.21
  4922.2  460.55  4932.9  460.16  4974.0  458.04  4984.3  458.15  4990.0  457.91
  4990.5  457.11  4995.5  457.11  4996.0  457.91  5004.8  457.99  5014.8  458.51
  5024.8  459.54  5029.0  460.16  5034.8  461.04  5064.8  460.92  5094.8  461.80
  5104.8  462.41  5114.8  463.28  5134.8  463.51  5224.8  465.79  5248.6  465.93
#Mann=3,-1,0
  4676.5    0.05       0  4990.0    0.03       0  4996.0    0.05       0
Bank Sta=4932.9,5029
Exp/Cntr=0.3,0.1

Type RM Length L Ch R = 1,11966,166,166,166
BEGIN DESCRIPTION:
XS3258A
END DESCRIPTION:
XS GIS Cut Line= 4
      2802222.81      7044238.68      2801916.41      7044186.79
      2801802.75      7044186.79      2801568.98      7044196.64
#Sta/Elev= 30
  4581.1  466.18  4609.3  465.07  4619.4  465.11  4670.2  463.40  4700.6  463.11
  4731.0  462.22  4752.1  462.00  4781.7  461.60  4802.0  460.88  4809.9  461.08
  4815.0  460.62  4862.9  460.26  4870.3  460.43  4875.4  459.84  4903.3  459.97
  4922.9  459.54  4963.3  457.96  4980.3  456.99  4980.8  456.19  4985.8  456.19
  4986.3  456.99  4993.3  457.75  5005.5  458.02  5029.7  459.54  5053.3  460.80
  5085.0  461.32  5103.4  462.49  5133.4  463.30  5203.4  464.13  5239.5  463.76
#Mann=4,-1,0
  4581.1    0.05       0  4752.1    0.08       0  4980.3    0.07       0
  4986.3    0.08       0
Bank Sta=4922.9,5029.7
Exp/Cntr=0.3,0.1

Type RM Length L Ch R = 1,11800,212,212,212
BEGIN DESCRIPTION:
XS3259A
END DESCRIPTION:
XS GIS Cut Line= 3
      2802274.69      7044080.54      2801909.00      7044083.01
      2801582.86      7044060.77
#Sta/Elev= 30
  4631.8  463.97  4634.1  463.97  4641.5  463.27  4651.5  463.01  4721.5  462.44
  4781.5  461.52  4801.5  461.36  4811.5  461.52  4831.5  460.56  4881.5  459.52
  4921.9  458.41  4971.5  457.52  4981.5  457.78  4991.5  457.41  4994.0  455.09
  4994.5  454.29  4999.5  454.29  5000.0  455.09  5011.5  455.42  5021.6  457.75
  5039.2  457.92  5044.2  457.68  5061.6  458.03  5104.9  458.41  5121.8  459.17
  5131.8  460.04  5232.0  460.86  5292.2  460.92  5312.2  461.39  5324.4  461.31
#Mann=3,-1,0
  4631.8    0.08       0  4994.0    0.07       0  5000.0    0.08       0
Bank Sta=4921.9,5104.9
Exp/Cntr=0.3,0.1

Type RM Length L Ch R = 1,11588,207,207,207
BEGIN DESCRIPTION:
XS3260A
END DESCRIPTION:
XS GIS Cut Line= 3
      2802200.60      7043944.64      2801928.77      7043872.97
      2801688.29      7043872.97
#Sta/Elev= 30
  4715.6  462.38  4762.8  461.97  4770.5  462.33  4775.6  462.24  4783.4  461.43
  4824.8  460.00  4845.5  459.53  4876.5  458.28  4884.4  457.16  4897.2  456.18
  4904.5  455.96  4905.0  455.16  4910.0  455.16  4910.5  455.96  4972.0  456.44
  4979.9  456.65  4990.3  456.48  4996.1  456.73  5010.5  456.70  5020.5  456.24
  5030.5  456.17  5050.5  456.78  5080.5  456.92  5090.5  457.26  5120.5  457.16
  5130.5  457.42  5140.5  458.60  5150.5  459.46  5220.5  459.87  5237.2  460.20
#Mann=3,-1,0
  4715.6    0.05       0  4904.5    0.03       0  4910.5    0.05       0
Bank Sta=4884.4,5120.5
Exp/Cntr=0.3,0.1

Type RM Length L Ch R = 1,11381,157,157,157
BEGIN DESCRIPTION:
XS3261A
END DESCRIPTION:
XS GIS Cut Line= 3
      2802167.36      7043756.19      2801950.39      7043669.39
      2801678.49      7043658.61
#Sta/Elev= 30
  4772.0  458.96  4784.3  459.01  4789.7  459.24  4796.1  458.69  4813.9  457.88
  4819.3  457.46  4828.4  457.08  4849.9  456.64  4867.8  457.31  4873.1  456.50
  4882.8  456.17  4921.6  455.84  4990.0  455.75  4999.7  453.58  5001.9  452.90
  5002.4  452.10  5007.4  452.10  5007.9  452.90  5011.1  455.53  5031.1  455.16
  5041.1  455.19  5061.1  455.43  5085.0  456.17  5141.2  458.28  5151.2  458.83
  5171.2  460.35  5221.2  461.04  5231.3  461.56  5251.3  461.77  5277.8  462.77
#Mann=3,-1,0
  4772.0    0.05       0  5001.9    0.03       0  5007.9    0.05       0
Bank Sta=4882.8,5085
Exp/Cntr=0.3,0.1

Type RM Length L Ch R = 1,11224,204,204,204
BEGIN DESCRIPTION:
XS3262A
END DESCRIPTION:
XS GIS Cut Line= 3
      2802226.04      7043647.72      2801985.11      7043517.49
      2801765.88      7043493.61
#Sta/Elev= 30
  4726.3  457.70  4737.8  457.70  4743.5  457.15  4759.7  457.51  4765.4  456.98
  4781.6  456.74  4825.4  455.63  4956.7  454.66  4988.9  454.78  4990.8  453.45
  4994.5  450.79  4995.0  449.99  5000.0  449.99  5000.5  450.79  5002.7  450.79
  5008.1  453.45  5010.3  454.51  5020.4  454.61  5030.5  454.06  5040.5  454.25
  5050.6  454.71  5072.5  454.95  5090.8  455.68  5100.9  455.69  5131.1  457.13
  5151.2  457.50  5158.9  458.31  5171.3  458.51  5191.4  459.95  5220.7  460.73
#Mann=3,-1,0
  4726.3    0.05       0  4994.5    0.03       0  5000.5    0.05       0
Bank Sta=4990.8,5008.1
Exp/Cntr=0.3,0.1

Type RM Length L Ch R = 1,11020,175,175,175
BEGIN DESCRIPTION:
XS3263A
END DESCRIPTION:
XS GIS Cut Line= 3
      2802234.69      7043315.66      2802004.64      7043324.34
      2801800.66      7043391.61
#Sta/Elev= 30
  4749.9  458.30  4779.6  457.75  4809.6  456.53  4869.8  455.24  4919.7  454.75
  4934.6  454.02  4969.7  453.65  4977.4  452.84  4982.6  452.84  4990.3  452.05
  4996.9  450.36  4999.1  449.42  4999.6  448.62  5004.6  448.62  5005.1  449.42
  5021.9  450.24  5028.6  452.82  5033.9  450.53  5042.9  450.48  5053.4  450.76
  5060.4  452.91  5065.6  450.62  5074.5  452.28  5083.8  453.17  5090.4  454.02
  5137.5  456.76  5155.6  458.75  5160.9  458.64  5187.4  460.43  5194.9  460.47
#Mann=5,-1,0
  4749.9    0.05       0  4999.1    0.03       0  5005.1    0.05       0
  5083.8    0.07       0  5137.5    0.05       0
Bank Sta=4934.6,5090.4
Exp/Cntr=0.3,0.1

Type RM Length L Ch R = 1,10845,116,116,116
BEGIN DESCRIPTION:
XS3264A
END DESCRIPTION:
XS GIS Cut Line= 3
      2802267.18      7043174.60      2801967.75      7043159.41
      2801785.50      7043174.60
#Sta/Elev= 30
  4706.5  460.30  4710.1  460.30  4728.7  458.60  4768.8  456.34  4795.6  455.89
  4800.6  455.42  4838.8  454.94  4874.1  453.87  4949.0  452.80  4979.0  452.96
  4989.0  451.46  4991.4  448.77  4991.9  447.97  4996.9  447.97  4997.4  448.77
  5005.2  451.22  5013.7  451.31  5019.1  452.71  5039.2  453.02  5069.3  451.82
  5079.3  452.50  5089.4  451.94  5099.4  452.38  5111.0  453.87  5115.5  454.40
  5129.1  456.19  5134.2  456.22  5139.5  457.95  5159.6  458.97  5189.2  458.40
#Mann=4,-1,0
  4706.5    0.05       0  4991.4    0.07       0  4997.4    0.05       0
  5115.5    0.05       0
Bank Sta=4874.1,5111
Exp/Cntr=0.3,0.1

Type RM Length L Ch R = 1,10729,196,196,196
BEGIN DESCRIPTION:
XS3265A
END DESCRIPTION:
XS GIS Cut Line= 3
      2802265.03      7043079.11      2802019.83      7043046.56
      2801815.89      7043040.06
#Sta/Elev= 30
  4726.1  459.08  4756.4  457.94  4766.5  457.90  4776.6  457.09  4793.5  456.75
  4798.6  456.96  4806.8  456.31  4827.0  455.85  4879.5  453.34  4940.1  452.23
  4945.2  452.05  4950.2  452.33  4973.4  450.68  4988.3  450.11  4995.3  448.27
  4995.8  447.47  5000.8  447.47  5001.3  448.27  5008.3  451.81  5018.3  452.25
  5038.3  452.56  5058.3  452.17  5078.3  452.66  5098.3  452.28  5108.4  451.43
  5114.7  452.23  5118.4  452.70  5131.4  455.34  5148.4  457.47  5177.5  457.19
#Mann=5,-1,0
  4726.1    0.05       0  4879.5    0.16       0  4995.3    0.07       0
  5001.3    0.16       0  5131.4    0.05       0
Bank Sta=4940.1,5114.7
Exp/Cntr=0.3,0.1

Type RM Length L Ch R = 1,10533,233,233,233
BEGIN DESCRIPTION:
XS3266A
END DESCRIPTION:
XS GIS Cut Line= 3
      2802171.78      7042799.15      2802011.15      7042870.78
      2801833.17      7042968.46
#Sta/Elev= 30
  4818.7  458.85  4859.0  457.35  4872.6  456.42  4895.9  453.72  4902.8  453.37
  4947.8  452.08  4957.5  452.83  4972.5  451.61  4979.4  451.18  4988.8  448.41
  4990.6  447.18  4991.1  446.38  4996.1  446.38  4996.6  447.18  5010.5  448.62
  5019.9  449.16  5038.0  450.28  5054.1  449.39  5059.8  450.27  5070.0  451.10
  5075.9  451.53  5081.6  451.37  5092.0  452.25  5097.7  451.48  5098.6  451.61
  5104.3  452.38  5135.6  454.04  5162.4  455.04  5179.2  456.42  5197.6  456.64
#Mann=5,-1,0
  4818.7    0.05       0  4990.6    0.03       0  4996.6    0.05       0
  5019.9    0.12       0  5162.4    0.05       0
Bank Sta=4972.5,5098.6
Exp/Cntr=0.3,0.1

Type RM Length L Ch R = 1,10300,164,164,164
BEGIN DESCRIPTION:
XS3267A
END DESCRIPTION:
XS GIS Cut Line= 3
      2802019.86      7042560.43      2801865.75      7042692.83
      2801759.72      7042926.53
#Sta/Elev= 30
  4805.1  456.54  4854.1  455.53  4939.1  451.14  4945.9  451.10  4960.5  450.00
  4989.0  449.77  4996.1  448.26  5000.3  445.90  5000.8  445.10  5005.8  445.10
  5006.3  445.90  5008.3  446.71  5012.2  446.71  5019.2  449.07  5024.7  449.88
  5032.6  450.28  5069.9  449.76  5109.5  450.16  5145.6  449.54  5153.4  449.93
  5158.5  451.14  5163.2  452.28  5168.6  451.36  5186.2  452.90  5191.7  452.49
  5197.3  453.75  5208.3  454.31  5214.8  454.61  5220.3  453.96  5264.9  456.06
#Mann=5,-1,0
  4805.1    0.05       0  4945.9    0.16       0  5000.3    0.07       0
  5006.3    0.16       0  5069.9    0.05       0
Bank Sta=4939.1,5158.5
Exp/Cntr=0.3,0.1

Type RM Length L Ch R = 1,10136,343,343,343
BEGIN DESCRIPTION:
XS3268A
END DESCRIPTION:
XS GIS Cut Line= 3
      2801804.99      7042425.90      2801744.22      7042595.18
      2801631.38      7042979.29
#Sta/Elev= 30
  4834.4  456.98  4886.6  453.56  4929.1  451.77  4942.2  450.71  4966.9  450.08
  4972.2  450.42  4992.3  448.57  4997.6  446.49  5000.4  444.65  5000.9  443.85
  5005.9  443.85  5006.4  444.65  5011.5  448.96  5034.9  449.23  5055.8  448.52
  5076.6  449.03  5107.9  448.58  5118.3  449.11  5138.0  449.28  5168.2  449.20
  5201.5  449.78  5206.8  449.50  5234.9  450.71  5240.1  451.03  5245.3  452.01
  5278.7  453.18  5345.5  454.06  5378.8  454.93  5399.7  455.93  5414.6  455.94
#Mann=4,-1,0
  4834.4    0.16       0  5000.4    0.07       0  5006.4    0.16       0
  5138.0    0.05       0
Bank Sta=4942.2,5234.9
Exp/Cntr=0.3,0.1

Type RM Length L Ch R = 1,9793,369,369,369
BEGIN DESCRIPTION:
XS3269A
END DESCRIPTION:
XS GIS Cut Line= 3
      2801689.96      7042326.09      2801561.93      7042471.48
      2801419.37      7042747.96
#Sta/Elev= 30
  4802.2  458.78  4812.3  458.56  4833.2  457.03  4875.9  453.25  4890.1  451.84
  4896.8  450.81  4904.4  450.34  4907.7  449.66  4911.0  448.98  4925.3  447.70
  4974.6  448.18  4982.2  447.93  4988.8  445.50  4991.9  443.13  4992.4  442.33
  4997.4  442.33  4997.9  443.13  5002.8  443.86  5011.1  447.00  5025.0  447.77
  5033.6  446.65  5041.5  447.73  5056.1  447.81  5078.6  449.05  5159.3  449.66
  5173.4  450.09  5218.8  451.47  5224.9  452.03  5235.4  452.36  5307.0  454.16
#Mann=4,-1,0
  4802.2    0.16       0  4991.9    0.07       0  4997.9    0.16       0
  5173.4    0.05       0
Bank Sta=4907.7,5159.3
Exp/Cntr=0.3,0.1

Type RM Length L Ch R = 1,9424,426,426,426
BEGIN DESCRIPTION:
UNT 047 in LFCCL Watershed 14.0
END DESCRIPTION:
XS GIS Cut Line= 3
      2801675.00      7042175.00      2801375.00      7042225.00
      2801064.97      7042501.86
#Sta/Elev= 30
  4734.6  460.07  4815.7  459.18  4889.2  455.45  4937.4  452.08  4945.0  450.54
  4949.0  448.27  4957.6  445.71  4988.1  446.55  4998.2  442.84  5002.8  442.38
  5003.3  441.58  5008.3  441.58  5008.8  442.38  5010.9  445.60  5018.5  447.03
  5028.6  446.72  5095.2  447.11  5131.1  446.72  5152.0  447.43  5187.1  447.62
  5199.6  448.27  5244.0  448.78  5251.5  449.19  5279.9  449.08  5335.9  449.95
  5392.8  451.88  5400.3  452.68  5407.6  452.74  5421.2  454.09  5454.4  455.63
#Mann=4,-1,0
  4734.6    0.16       0  5002.8    0.07       0  5008.8    0.16       0
  5407.6    0.05       0
Bank Sta=4949,5199.6
Exp/Cntr=0.3,0.1

Type RM Length L Ch R = 1,8998,380,380,380
BEGIN DESCRIPTION:
UNT 047 in LFCCL Watershed 13.0
END DESCRIPTION:
XS GIS Cut Line= 3
      2801525.01      7041925.00      2801225.00      7041925.00
      2800775.01      7042524.99
#Sta/Elev= 30
  4725.0  459.25  4765.0  458.21  4808.9  455.25  4816.9  454.52  4855.0  451.28
  4875.0  447.82  4890.1  446.20  4915.0  445.03  4956.1  445.77  4975.0  445.82
  4985.0  445.03  5002.0  441.25  5002.5  440.45  5007.5  440.45  5008.0  441.25
  5015.0  441.93  5022.5  444.44  5032.3  443.70  5076.9  446.07  5097.0  446.20
  5098.1  446.21  5111.5  446.79  5246.9  446.81  5353.1  448.65  5495.6  453.90
  5578.7  457.08  5588.2  457.63  5746.9  464.52  5767.7  464.58  5775.0  465.42
#Mann=11,-1,0
  4725.0    0.05       0  4808.9    0.16       0  4816.9    0.05       0
  4956.1    0.16       0  5002.0    0.07       0  5008.0    0.16       0
  5076.9    0.07       0  5098.1    0.16       0  5495.6    0.05       0
  5578.7    0.08       0  5588.2    0.05       0
Bank Sta=4890.1,5097
Exp/Cntr=0.3,0.1

Type RM Length L Ch R = 1,8618,322,322,322
BEGIN DESCRIPTION:
UNT 047 in LFCCL Watershed 12.0
END DESCRIPTION:
XS GIS Cut Line= 3
      2801524.98      7041475.01      2801225.00      7041575.00
      2800775.00      7042025.00
#Sta/Elev= 30
  4700.0  456.65  4742.1  455.37  4752.7  454.41  4805.4  453.44  4815.9  452.51
  4837.0  451.86  4847.6  450.83  4900.3  448.07  4910.8  446.73  4931.9  445.16
  4953.9  444.18  4995.1  442.97  5002.7  440.56  5003.2  439.76  5008.2  439.76
  5008.7  440.56  5013.6  443.59  5058.6  443.21  5115.2  444.98  5129.3  444.25
  5157.6  444.56  5171.8  444.18  5185.9  442.57  5214.2  443.98  5242.5  443.72
  5256.6  442.94  5292.5  444.18  5454.6  448.58  5553.6  452.59  5652.6  455.97
#Mann=3,-1,0
  4700.0    0.05       0  5002.7    0.03       0  5008.7    0.05       0
Bank Sta=4953.9,5292.5
Exp/Cntr=0.3,0.1

Type RM Length L Ch R = 1,8296,475,475,475
BEGIN DESCRIPTION:
XS3270A
END DESCRIPTION:
XS GIS Cut Line= 3
      2801375.26      7041241.02      2801043.27      7041329.99
      2800863.15      7041453.68
#Sta/Elev= 30
  4666.5  455.75  4734.6  453.72  4777.0  451.32  4811.7  450.33  4817.0  449.39
  4822.2  449.34  4880.8  443.31  4897.0  441.62  4937.1  442.89  4966.7  442.51
  4977.3  443.40  4998.1  442.06  5003.7  439.98  5004.2  439.18  5009.2  439.18
  5009.7  439.98  5010.2  440.97  5020.2  441.98  5063.0  443.31  5083.9  443.30
  5105.1  441.96  5141.5  442.25  5155.6  440.30  5170.5  441.74  5177.9  442.97
  5192.2  443.31  5200.3  444.73  5206.4  445.16  5221.3  448.67  5228.7  448.96
#Mann=4,-1,0
  4666.5    0.08       0  4734.6    0.05       0  5003.7    0.03       0
  5009.7    0.05       0
Bank Sta=4880.8,5192.2
Exp/Cntr=0.3,0.1

Type RM Length L Ch R = 1,7821,406,406,406
BEGIN DESCRIPTION:
XS3271A
END DESCRIPTION:
XS GIS Cut Line= 3
      2801292.84      7041045.70      2800804.55      7041186.76
      2800672.21      7041338.63
#Sta/Elev= 30
  4501.2  449.94  4593.3  446.98  4660.6  443.96  4665.8  444.43  4700.7  442.54
  4766.6  441.65  4805.5  441.98  4821.6  441.03  4852.9  440.62  4872.7  441.96
  4894.5  442.13  4984.0  441.16  4995.6  437.72  4996.1  436.92  5001.1  436.92
  5001.6  437.72  5006.6  439.40  5011.6  439.40  5015.1  441.38  5021.7  440.46
  5043.6  441.67  5047.9  442.54  5064.4  443.76  5072.0  445.15  5078.7  447.85
  5086.3  448.25  5113.8  447.01  5170.8  449.14  5178.4  448.27  5210.9  449.23
#Mann=3,-1,0
  4501.2    0.05       0  4995.6    0.03       0  5001.6    0.05       0
Bank Sta=4700.7,5047.9
Exp/Cntr=0.3,0.1

Type RM Length L Ch R = 1,7415,544,544,544
BEGIN DESCRIPTION:
UNT 047 in LFCCL Watershed 11.0
END DESCRIPTION:
XS GIS Cut Line= 3
      2801375.04      7040925.01      2800775.00      7040825.00
      2800539.90      7040763.61
#Sta/Elev= 30
  4386.4  454.35  4447.3  450.26  4457.4  450.20  4487.8  447.83  4528.4  446.90
  4548.6  444.74  4568.9  444.77  4624.5  441.77  4690.6  440.47  4741.3  441.19
  4779.3  440.17  4784.4  440.85  4795.4  439.67  4812.2  439.17  4840.1  440.02
  4845.2  439.29  4883.2  440.55  4933.9  440.26  4954.2  440.94  4997.3  439.66
  5002.0  437.24  5002.5  436.44  5007.6  436.44  5008.1  437.24  5011.6  441.76
  5012.2  442.59  5017.5  444.93  5139.4  453.71  5201.4  454.79  5237.7  456.28
#Mann=5,-1,0
  4386.4    0.05       0  4795.4    0.16       0  5002.0    0.07       0
  5008.1    0.16       0  5012.2    0.05       0
Bank Sta=4624.5,5011.6
Exp/Cntr=0.3,0.1

Type RM Length L Ch R = 1,6871,570,570,570
BEGIN DESCRIPTION:
UNT 047 in LFCCL Watershed 10.0
END DESCRIPTION:
XS GIS Cut Line= 3
      2801475.00      7040775.00      2801075.00      7040425.00
      2800624.97      7040475.00
#Sta/Elev= 30
  4429.4  455.34  4535.7  450.83  4571.3  448.22  4614.0  447.05  4649.1  444.15
  4684.2  443.73  4706.1  442.00  4760.3  440.26  4769.7  439.33  4826.6  439.63
  4854.6  437.96  4921.2  438.87  4925.3  438.96  4932.9  436.84  4939.6  436.84
  4947.1  438.95  4971.0  438.64  4988.0  436.26  4988.5  435.46  4993.6  435.46
  4994.1  436.26  5001.2  438.62  5021.3  439.41  5071.6  437.95  5138.9  440.26
  5152.1  441.41  5182.3  448.93  5204.0  452.62  5313.1  455.88  5413.7  455.60
#Mann=5,-1,0
  4429.4    0.05       0  4921.2    0.16       0  4988.0    0.07       0
  4994.1    0.16       0  5204.0    0.05       0
Bank Sta=4760.3,5138.9
Exp/Cntr=0.3,0.1

Type RM Length L Ch R = 1,6301,412,412,412
BEGIN DESCRIPTION:
UNT 047 in LFCCL Watershed 9.0
END DESCRIPTION:
XS GIS Cut Line= 3
      2801775.05      7040025.01      2801325.00      7039975.00
      2800625.01      7040125.00
#Sta/Elev= 30
  4529.6  453.23  4559.8  452.62  4650.4  448.56  4700.7  444.05  4781.2  439.94
  4814.6  439.00  4851.6  437.57  4874.4  437.52  4901.9  436.70  4932.1  437.09
  4942.2  437.89  4962.3  437.06  4972.4  437.78  4992.6  436.79  5002.0  437.73
  5004.1  436.58  5004.6  435.78  5009.7  435.78  5010.2  436.58  5013.1  437.86
  5023.3  437.96  5150.3  437.53  5170.8  436.69  5219.8  437.51  5272.6  437.92
  5313.3  439.00  5452.9  442.40  5530.4  446.71  5565.4  447.64  5698.3  453.79
#Mann=7,-1,0
  4529.6    0.05       0  4874.4    0.12       0  5004.1    0.07       0
  5010.2    0.12       0  5170.8    0.16       0  5219.8     0.1       0
  5272.6    0.05       0
Bank Sta=4814.6,5313.3
Exp/Cntr=0.3,0.1

Type RM Length L Ch R = 1,5889,402,402,402
BEGIN DESCRIPTION:
XS3272A
END DESCRIPTION:
XS GIS Cut Line= 3
      2801688.68      7039806.12      2801414.36      7039740.14
      2800921.36      7039781.80
#Sta/Elev= 30
  4718.3  447.87  4746.1  446.76  4767.1  445.35  4830.0  442.66  4835.2  442.09
  4845.5  442.15  4868.4  441.39  4938.1  439.03  4949.0  437.96  4955.9  436.48
  4968.9  435.36  4979.2  435.84  4994.4  434.32  4994.9  433.52  5000.1  433.52
  5000.6  434.32  5002.6  434.32  5009.8  436.39  5070.0  436.28  5150.3  436.83
  5210.5  436.24  5220.6  435.34  5250.7  436.32  5269.0  436.31  5310.9  437.41
  5350.5  438.11  5355.5  437.61  5361.5  437.96  5431.3  440.72  5495.2  444.62
#Mann=6,-1,0
  4718.3    0.16       0  4767.1    0.05       0  4868.4    0.12       0
  4994.4    0.07       0  5000.6    0.12       0  5269.0    0.16       0
Bank Sta=4949,5361.5
Exp/Cntr=0.3,0.1

Type RM Length L Ch R = 1,5487,663,663,663
BEGIN DESCRIPTION:
UNT 047 in LFCCL Watershed 8.0
END DESCRIPTION:
XS GIS Cut Line= 3
      2801924.98      7039538.89      2801475.00      7039488.89
      2800875.05      7039488.89
#Sta/Elev= 30
  4595.4  453.93  4673.4  454.43  4696.0  452.55  4706.1  452.39  4746.3  453.30
  4753.5  451.90  4763.9  450.39  4796.6  448.97  4854.5  444.92  4930.4  441.13
  4977.7  439.85  4987.8  436.91  4997.8  434.01  5007.9  435.68  5018.0  435.71
  5108.1  435.44  5158.1  434.71  5178.1  435.11  5185.0  433.95  5185.5  433.15
  5190.7  433.15  5191.2  433.95  5208.1  434.99  5298.1  434.55  5363.7  436.91
  5418.1  439.37  5475.6  442.99  5498.1  444.76  5558.1  448.15  5648.1  451.21
#Mann=6,-1,0
  4595.4    0.05       0  4753.5    0.16       0  4930.4    0.12       0
  5185.0    0.07       0  5191.2    0.12       0  5475.6    0.16       0
Bank Sta=4987.8,5363.7
Exp/Cntr=0.3,0.1

Type RM Length L Ch R = 1,4824,204,204,204
BEGIN DESCRIPTION:
UNT 047 in LFCCL Watershed 7.0
END DESCRIPTION:
XS GIS Cut Line= 3
      2801774.98      7039125.00      2801325.00      7039125.00
      2800875.01      7039424.99
#Sta/Elev= 30
  4520.5  450.86  4568.7  448.99  4646.7  445.29  4720.5  441.95  4750.5  435.48
  4756.7  434.83  4810.5  434.77  4850.5  433.77  4930.5  434.05  4960.5  432.99
  4968.0  433.71  4984.0  433.44  4993.0  427.11  4999.0  427.61  5003.4  425.85
  5003.9  425.05  5009.1  425.05  5009.6  425.85  5014.0  433.50  5020.1  432.81
  5029.1  433.99  5065.1  433.40  5071.1  434.30  5092.2  434.89  5143.2  434.28
  5173.5  434.80  5174.8  434.83  5209.3  435.22  5410.7  447.50  5511.3  451.35
#Mann=6,-1,0
  4520.5    0.05       0  4568.7    0.16       0  4646.7    0.12       0
  5003.4    0.07       0  5009.6    0.12       0  5173.5    0.16       0
Bank Sta=4756.7,5174.8
Exp/Cntr=0.3,0.1

Type RM Length L Ch R = 1,4620,356,356,356
BEGIN DESCRIPTION:
XS3275A
END DESCRIPTION:
XS GIS Cut Line= 3
      2801558.43      7038962.36      2801240.75      7038957.16
      2800908.76      7039019.40
#Sta/Elev= 30
  4762.1  440.12  4766.3  440.12  4775.5  439.11  4795.5  438.05  4825.5  435.26
  4855.5  434.31  4865.1  433.59  4925.6  433.50  4945.6  433.16  4955.6  433.41
  4975.6  433.07  4985.6  431.69  4995.6  426.74  5002.5  424.87  5003.0  424.07
  5008.2  424.07  5008.7  424.87  5025.6  433.02  5065.6  433.47  5093.0  433.17
  5145.6  433.27  5171.7  433.59  5208.3  434.24  5248.5  434.40  5279.0  435.27
  5308.4  435.70  5329.9  436.26  5382.2  438.36  5401.1  439.27  5417.6  440.53
#Mann=4,-1,0
  4762.1    0.12       0  5002.5    0.07       0  5008.7    0.12       0
  5382.2    0.16       0
Bank Sta=4865.1,5171.7
Exp/Cntr=0.3,0.1

Type RM Length L Ch R = 1,4264,687,687,687
BEGIN DESCRIPTION:
UNT 047 in LFCCL Watershed 6.0
END DESCRIPTION:
XS GIS Cut Line= 3
      2801675.00      7038925.00      2801325.00      7038625.00
      2800874.95      7038574.99
#Sta/Elev= 30
  4543.7  448.78  4550.8  449.45  4560.8  448.58  4565.1  448.42  4571.7  446.33
  4593.6  444.37  4614.5  444.12  4639.3  441.87  4688.7  439.84  4714.4  436.95
  4721.0  438.47  4728.1  438.62  4792.3  434.09  4866.8  432.00  4969.0  431.92
  4976.7  427.88  4983.3  429.42  4991.0  423.89  4994.4  423.11  4994.9  422.31
  5000.2  422.31  5000.7  423.11  5001.4  425.51  5007.2  425.51  5014.7  429.90
  5024.8  431.96  5051.8  432.00  5183.2  434.14  5316.6  438.70  5457.5  445.55
#Mann=7,-1,0
  4543.7    0.16       0  4560.8    0.12       0  4639.3    0.16       0
  4688.7    0.12       0  4994.4    0.07       0  5000.7    0.12       0
  5183.2    0.16       0
Bank Sta=4866.8,5051.8
Exp/Cntr=0.3,0.1

Type RM Length L Ch R = 1,3577,585,585,585
BEGIN DESCRIPTION:
UNT 047 in LFCCL Watershed 5.0
END DESCRIPTION:
XS GIS Cut Line= 3
      2801875.00      7038525.00      2801475.00      7038175.00
      2800824.95      7038074.99
#Sta/Elev= 30
  4488.6  446.39  4491.8  446.39  4524.2  445.41  4530.8  442.48  4552.7  440.24
  4573.5  442.14  4736.8  433.77  4867.5  430.24  4893.6  429.74  4920.9  429.93
  4935.2  426.40  4956.0  429.73  4977.9  427.46  4984.5  428.54  4986.9  424.63
  4992.1  420.71  5006.3  422.00  5009.8  420.39  5010.3  419.59  5016.1  420.39
  5016.8  428.20  5030.2  429.92  5047.4  429.45  5132.7  429.74  5173.6  431.09
  5262.9  433.85  5283.2  435.74  5303.4  432.70  5323.6  436.48  5677.8  452.28
#Mann=7,-1,0
  4488.6    0.16       0  4491.8    0.05       0  4867.5    0.16       0
  5009.8    0.07       0  5016.1    0.16       0  5047.4    0.12       0
  5173.6    0.16       0
Bank Sta=4893.6,5132.7
Exp/Cntr=0.3,0.1

Type RM Length L Ch R = 1,2992,528,528,528
BEGIN DESCRIPTION:
UNT 047 in LFCCL Watershed 4.0
END DESCRIPTION:
XS GIS Cut Line= 3
      2801925.04      7037374.97      2801575.00      7037675.00
      2800875.03      7037924.99
#Sta/Elev= 30
  4554.6  449.07  4596.4  446.43  4726.3  438.24  4750.9  436.19  4781.3  432.89
  4859.2  429.60  4929.5  428.55  4949.8  428.09  4965.7  427.65  4973.4  422.13
  4987.6  420.24  4994.2  421.83  4998.4  418.80  4998.9  418.00  5004.9  418.00
  5005.4  418.80  5008.5  418.84  5012.3  425.59  5018.3  425.59  5025.7  427.93
  5111.2  427.19  5154.2  427.90  5196.1  424.41  5210.5  426.93  5241.3  427.87
  5259.9  425.28  5270.1  428.55  5281.1  432.57  5379.7  436.31  5758.9  451.33
#Mann=8,-1,0
  4554.6    0.05       0  4596.4    0.16       0  4726.3    0.12       0
  4750.9    0.16       0  4949.8    0.12       0  4998.4    0.07       0
  5005.4    0.12       0  5379.7    0.16       0
Bank Sta=4929.5,5270.1
Exp/Cntr=0.3,0.1

Type RM Length L Ch R = 1,2464,750,750,750
BEGIN DESCRIPTION:
UNT 047 in LFCCL Watershed 3.0
END DESCRIPTION:
XS GIS Cut Line= 3
      2801575.00      7037025.00      2801225.00      7037325.00
      2800924.98      7037725.02
#Sta/Elev= 30
  4570.7  444.24  4577.8  444.90  4606.4  434.65  4613.0  433.71  4666.6  432.02
  4684.6  431.55  4748.0  429.63  4764.9  430.29  4840.1  429.16  4891.6  426.74
  4925.8  423.93  4939.5  426.53  4953.2  424.96  4960.9  426.58  4981.7  427.14
  4989.4  424.26  4996.0  418.09  5000.1  417.40  5000.7  416.60  5007.2  417.40
  5010.3  421.20  5024.5  426.75  5068.1  426.75  5103.5  424.44  5136.2  426.74
  5181.7  427.56  5266.7  432.52  5271.3  432.88  5382.9  439.13  5531.7  445.54
#Mann=9,-1,0
  4570.7    0.16       0  4666.6    0.12       0  4684.6    0.16       0
  4764.9    0.12       0  5000.1    0.07       0  5007.2    0.12       0
  5266.7    0.16       0  5271.3    0.12       0  5382.9    0.16       0
Bank Sta=4891.6,5136.2
Exp/Cntr=0.3,0.1

Type RM Length L Ch R = 1,1714,614,614,614
BEGIN DESCRIPTION:
UNT 047 in LFCCL Watershed 2.0
END DESCRIPTION:
XS GIS Cut Line= 3
      2801025.00      7036575.00      2800975.00      7037025.00
      2800625.00      7037525.00
#Sta/Elev= 30
  4475.4  451.44  4489.8  451.42  4606.2  448.64  4687.1  443.60  4817.5  432.86
  4857.7  427.19  4882.8  425.77  4898.0  421.28  4908.0  423.56  4918.1  417.35
  4935.6  416.52  4941.7  417.56  4956.5  417.03  4964.8  422.44  4971.3  423.98
  4986.2  424.80  4992.3  422.69  5001.0  422.83  5007.1  417.39  5010.1  416.44
  5010.6  415.64  5017.2  416.44  5021.9  416.66  5036.7  424.56  5047.8  425.77
  5139.8  427.51  5216.9  428.68  5251.2  429.26  5358.4  434.67  5538.5  443.78
#Mann=8,-1,0
  4475.4    0.05       0  4489.8    0.16       0  4687.1    0.12       0
  5010.1    0.07       0  5017.2    0.12       0  5139.8    0.16       0
  5216.9    0.12       0  5358.4    0.16       0
Bank Sta=4882.8,5047.8
Exp/Cntr=0.3,0.1

Type RM Length L Ch R = 1,1100,875,875,875
BEGIN DESCRIPTION:
XS3273A
END DESCRIPTION:
XS GIS Cut Line= 3
      2800681.72      7036570.03      2800660.89      7036941.53
      2800480.34      7037465.83
#Sta/Elev= 30
  4626.4  449.50  4656.8  446.40  4661.8  447.01  4681.5  444.10  4721.5  436.68
  4761.6  427.05  4778.4  424.92  4891.8  424.70  4901.8  423.91  4911.8  421.00
  4921.8  420.75  4951.9  424.00  4971.9  422.04  4981.9  423.37  4991.9  421.08
  4994.2  415.03  4994.7  414.23  5001.3  415.03  5004.3  416.17  5012.7  415.30
  5030.3  423.73  5035.6  422.57  5044.5  425.05  5098.0  423.53  5118.5  425.17
  5165.6  424.92  5278.9  427.47  5369.1  432.26  5419.9  435.07  5553.0  444.07
#Mann=6,-1,0
  4626.4    0.12       0  4994.2    0.07       0  5001.3    0.12       0
  5278.9    0.16       0  5369.1    0.12       0  5419.9    0.16       0
Bank Sta=4778.4,5165.6
Exp/Cntr=0.3,0.1

Type RM Length L Ch R = 1,225,0,0,0
BEGIN DESCRIPTION:
UNT 047 in LFCCL Watershed 1.0
END DESCRIPTION:
XS GIS Cut Line= 3
      2800496.56      7036429.97      2800246.55      7036829.98
      2800196.55      7037429.99
#Sta/Elev= 30
  4520.6  441.60  4721.4  435.63  4794.5  429.37  4815.7  428.37  4836.9  429.46
  4873.5  427.52  4888.8  425.19  4894.7  425.69  4905.5  422.01  4910.1  420.28
  4931.3  420.26  4946.6  422.34  4974.6  422.63  4983.2  416.64  4992.3  416.03
  4993.8  413.52  4994.3  412.72  5000.9  413.52  5007.4  413.93  5017.4  421.55
  5047.5  423.09  5057.6  421.08  5066.9  417.29  5071.9  420.44  5078.0  422.01
  5087.7  423.30  5248.2  423.43  5380.2  426.43  5569.3  435.42  5594.4  434.86
#Mann=4,-1,0
  4520.6    0.12       0  4993.8    0.07       0  5000.9    0.12       0
  5380.2    0.16       0
Bank Sta=4905.5,5078
Exp/Cntr=0.3,0.1

Chan Stop Cuts=-1
